--- WEST CANEY CREEK.prj (project) ---

Proj Title=WEST CANEY CREEK Base Level Engineering
Current Plan=p01
Default Exp/Contr=0.3,0.1
English Units
Geom File=g01
Flow File=f01
Plan File=p01
Y Axis Title=Elevation
X Axis Title(PF)=Main Channel Distance
X Axis Title(XS)=Station
BEGIN DESCRIPTION:
WEST CANEY CREEK
END DESCRIPTION:
DSS Export Rating Curves= 0
DSS Export Rating Curve Sorted= 0
DSS Export Volume Flow Curves= 0
DXF OffsetX= 0
DXF OffsetY= 0
DXF ScaleX= 1
DXF ScaleY= 10

--- WEST CANEY CREEK.p01 (plan) ---

Plan Title=Multiple Run
Short Identifier=Multiple
Geom File=g01
Flow File=f01
Subcritical Flow
K Sum by GR= 0
Std Step Tol= 0.01
Critical Tol= 0.01
Num of Std Step Trials= 20
Max Error Tol= 0.3
Flow Tol Ratio= 0.001
Split Flow NTrial= 30
Split Flow Tol= 0.02
Split Flow Ratio= 0.02
Log Output Level= 0
Friction Slope Method= 1
Unsteady Friction Slope Method= 2
Unsteady Bridges Friction Slope Method= 1
Parabolic Critical Depth
Global Vel Dist=  1 , 1 , 1
Global Log Level= 0
CheckData=True
Encroach Param= -1, 0, 0, 0
BEGIN DESCRIPTION:
Multiple Run
END DESCRIPTION:

--- WEST CANEY CREEK.f01 (steady flow) ---

Flow Title=Multiple
Program Version=4.10
Number of Profiles= 7
Profile Names=10-year,25-year,50-year,1pct_min,100-year,1pct_plu,500-year
River Rch & RM=WEST CANEY CREEK,Reach-1         ,64757
    1124    1538    1878    1672    2261    3058    3267
River Rch & RM=WEST CANEY CREEK,Reach-1         ,56602
    2176    3082    3852    3502    4736    6405    7142
River Rch & RM=WEST CANEY CREEK,Reach-1         ,53747
    2176    3082    3852    3502    4736    6405    7142
River Rch & RM=WEST CANEY CREEK,Reach-1         ,51425
    2428    3457    4334    3952    5344    7228    8108
River Rch & RM=WEST CANEY CREEK,Reach-1         ,49717
    2735    3918    4935    4521    6114    8268    9369
River Rch & RM=WEST CANEY CREEK,Reach-1         ,46749
    2791    3999    5035    4613    6238    8436    9567
River Rch & RM=WEST CANEY CREEK,Reach-1         ,41367
    5707    8441   10865   10155   13734   18573   21914
River Rch & RM=WEST CANEY CREEK,Reach-1         ,40472
    5707    8441   10865   10155   13734   18573   21914
River Rch & RM=WEST CANEY CREEK,Reach-1         ,35033
    6793   10093   13031   12213   16516   22337   26494
River Rch & RM=WEST CANEY CREEK,Reach-1         ,33794
    6793   10093   13031   12213   16516   22337   26494
River Rch & RM=WEST CANEY CREEK,Reach-1         ,28791
    6907   10258   13240   12406   16777   22689   26903
River Rch & RM=WEST CANEY CREEK,Reach-1         ,24691
    6867   10166   13093   12242   16556   22391   26448
River Rch & RM=WEST CANEY CREEK,Reach-1         ,18937
    7716   11453   14780   13847   18726   25325   30041
River Rch & RM=WEST CANEY CREEK,Reach-1         ,13985
    7716   11453   14780   13847   18726   25325   30041
River Rch & RM=WEST CANEY CREEK,Reach-1         ,7021
    7661   11342   14611   13664   18479   24991   29546
River Rch & RM=WEST CANEY CREEK,Reach-1         ,4841
    7661   11342   14611   13664   18479   24991   29546
Boundary for River Rch & Prof#=WEST CANEY CREEK,Reach-1         , 1
Up Type= 0
Dn Type= 3
Dn Slope=0.00116
Boundary for River Rch & Prof#=WEST CANEY CREEK,Reach-1         , 2
Up Type= 0
Dn Type= 3
Dn Slope=0.00116
Boundary for River Rch & Prof#=WEST CANEY CREEK,Reach-1         , 3
Up Type= 0
Dn Type= 3
Dn Slope=0.00116
Boundary for River Rch & Prof#=WEST CANEY CREEK,Reach-1         , 4
Up Type= 0
Dn Type= 3
Dn Slope=0.00116
Boundary for River Rch & Prof#=WEST CANEY CREEK,Reach-1         , 5
Up Type= 0
Dn Type= 3
Dn Slope=0.00116
Boundary for River Rch & Prof#=WEST CANEY CREEK,Reach-1         , 6
Up Type= 0
Dn Type= 3
Dn Slope=0.00116
Boundary for River Rch & Prof#=WEST CANEY CREEK,Reach-1         , 7
Up Type= 0
Dn Type= 3
Dn Slope=0.00116
DSS Import GetInterval= 0
DSS Import GetPeak= 0
DSS Import FillOption= 0

--- WEST CANEY CREEK.g01 (geometry) ---

Geom Title=Existing Conditions
Program Version=4.10

River Reach=WEST CANEY CREEK,Reach-1
Reach XY= 30
      3612746.01     10360733.52      3613312.97      10359845.7
      3612992.22     10358876.95        3613714.     10356147.33
       3614288.5     10355956.92      3613738.71     10353887.22
      3610439.13     10352119.42      3609857.47     10350284.53
      3609126.61       10350411.      3607212.17      10347864.9
      3607346.72      10347367.5      3606402.56     10347361.86
      3606417.06     10346329.09      3604736.59     10344349.48
      3603653.65     10345078.27      3603244.74     10343656.53
      3599473.51     10342958.58      3598972.17     10341970.33
      3597168.63     10341288.49      3597231.85     10340772.87
      3596533.09      10340570.4      3596574.99     10339226.73
      3594704.44     10339561.95      3592515.56     10336840.28
      3592549.63     10334892.67      3590717.02     10333734.55
      3590601.84     10333292.05      3591300.16     10333286.11
      3591069.76     10332502.56      3589772.11     10331261.64

Type RM Length L Ch R = 1 ,64757   ,442,442,442
BEGIN DESCRIPTION:
WEST CANEY CREEK 75.0
END DESCRIPTION:
XS GIS Cut Line= 3
      3613468.51     10360890.27      3613049.02     10360579.84
       3612386.7     10360051.66
#Sta/Elev= 30
  4339.4  379.66    4385  379.04  4449.7  376.97  4471.8  377.06  4499.8   376.1
  4535.3   375.8  4608.4  372.84  4621.1  372.87  4650.1  370.98    4694  369.99
  4714.8  368.54  4779.6  366.51    4928  363.88  4972.3  364.55  4985.2  363.88
  4990.2   362.4  4992.9   361.9  4996.2   362.4    5022  363.65  5028.4  363.14
  5036.4  363.69  5075.3  364.17  5177.3  363.41  5228.2  365.44  5476.8  370.46
  5584.1   375.1  5668.9  376.12  5689.7  376.91  5697.7  378.09  5708.4  378.02
#Mann= 5 ,-1 , 0
  4339.4     .05       0    4928     .16       0  4990.2     .07       0
  4996.2     .16       0  5075.3     .05       0
Bank Sta=4985.2,5022
XS Rating Curve= 0 ,0
Exp/Cntr=0.3,0.1

Type RM Length L Ch R = 1 ,64315   ,1240,1240,1240
BEGIN DESCRIPTION:
WEST CANEY CREEK 74.0
END DESCRIPTION:
XS GIS Cut Line= 3
       3613762.1     10360344.91      3613426.55     10360244.25
      3612461.77     10359908.67
#Sta/Elev= 30
  4329.3  375.88  4494.2  374.48  4565.5  372.51  4570.8   372.9  4579.9  372.11
  4611.2  371.35    4769  364.76  4849.1  363.12  4874.9  362.08  4919.2   362.1
    4945  361.25  4981.4  361.82  4998.9  358.46  5001.7  357.96  5004.9  358.46
  5012.5  361.03  5023.1  361.66  5074.2   361.9  5126.3  363.05  5162.7  362.93
  5188.5  364.06  5234.9  364.56  5276.5  365.92    5344  366.36  5369.8  367.16
  5375.1  366.78  5449.5   368.9  5499.9  369.47  5573.7   370.9  5701.1  376.08
#Mann= 7 ,-1 , 0
  4329.3     .05       0  4849.1     .16       0  4998.9     .07       0
  5004.9     .16       0  5074.2     .05       0  5449.5     .16       0
  5499.9     .05       0
Bank Sta=4981.4,5023.1
XS Rating Curve= 0 ,0
Exp/Cntr=0.3,0.1

Type RM Length L Ch R = 1 ,63075   ,1369,1369,1369
BEGIN DESCRIPTION:
WEST CANEY CREEK 73.0
END DESCRIPTION:
XS GIS Cut Line= 3
      3613963.53     10359942.25      3613544.01     10359564.68
       3612428.2     10359589.85
#Sta/Elev= 30
  4202.7  370.23  4515.4  369.59  4621.7  368.12  4635.8  369.25  4657.4  369.83
  4678.4  368.24  4685.8  368.28    4700  366.88  4749.4  366.62  4763.6  365.53
  4770.6  365.99    4839     363  4909.9  362.11  4969.1  358.78  4996.1  353.78
  4998.8  353.28  5002.1  353.78  5009.1  354.65  5019.1  356.99  5029.1  357.91
  5058.4  358.42  5199.1  359.63  5247.3  360.65  5300.7  361.68  5359.2  361.72
  5429.2  362.71  5569.2  365.82  5719.3  372.21  5792.6  374.42  5883.2  377.06
#Mann= 7 ,-1 , 0
  4202.7     .05       0  4909.9     .16       0  4996.1     .07       0
  5002.1     .16       0  5058.4     .05       0  5247.3     .16       0
  5792.6     .05       0
Bank Sta=4969.1,5029.1
XS Rating Curve= 0 ,0
Exp/Cntr=0.3,0.1

Type RM Length L Ch R = 1 ,61706   ,151,151,151
BEGIN DESCRIPTION:
WEST CANEY CREEK 72.0
END DESCRIPTION:
XS GIS Cut Line= 3
      3613996.47     10359432.66      3612619.72     10358514.25
      3612368.03     10358488.22
#Sta/Elev= 30
  3931.4  367.92    3955  367.67  4245.9   364.9  4291.3  365.25  4302.2  365.14
    4339  365.31  4479.3  362.41  4533.7  361.27  4855.2  357.63  4880.9  356.55
  4951.9  355.74  4966.9  353.98  4981.9  351.57  4987.9  349.53  4991.5  349.45
  4994.2  348.95  4997.5  349.45    5018  351.45    5024  353.24    5039  353.13
  5043.2  355.53    5045  356.56  5075.1   358.8  5198.2   361.5  5575.3  363.55
  5734.8  366.32  5753.7  365.72    5785   366.9  5825.2  366.82  5839.4  367.66
#Mann= 12 ,-1 , 0
  3931.4     .08       0    3955     .05       0  4291.3     .08       0
  4302.2     .05       0  4479.3     .08       0  4533.7     .05       0
  4855.2     .08       0  4880.9     .05       0  4991.5     .07       0
  4997.5     .05       0  5043.2     .05       0  5575.3      .1       0
Bank Sta=4951.9,5043.2
XS Rating Curve= 0 ,0
Exp/Cntr=0.3,0.1

Type RM Length L Ch R = 1 ,61555   ,648,648,648
BEGIN DESCRIPTION:
WEST CANEY CREEK 71.0
END DESCRIPTION:
XS GIS Cut Line= 3
      3613949.55     10359264.23      3612626.66     10358312.86
      3612556.27     10358292.26
#Sta/Elev= 30
  4047.8  364.99  4086.6  364.64  4126.2   364.5  4264.5  364.79  4313.6  365.34
  4334.5  364.42  4363.9  365.46  4412.8  363.81  4577.6  360.16  4717.9  358.51
    4798     357  4836.3  355.77  4900.4  355.02  4929.8  357.69  4971.6  354.87
  4975.9  354.04  4986.3  352.25  4990.1  349.84  4992.8  349.34  4996.1  349.84
  5007.2  350.31  5036.6  354.98    5073  356.33  5153.7  357.95  5191.3  358.21
  5288.3  360.26  5331.6  359.64    5477  361.24  5645.6  361.86  5750.6  364.19
#Mann= 18 ,-1 , 0
  4047.8     .08       0  4086.6     .05       0  4126.2     .08       0
  4264.5     .05       0  4412.8     .08       0  4577.6     .05       0
  4717.9     .08       0    4798     .12       0  4836.3     .08       0
  4975.9     .05       0  4990.1     .03       0  4996.1     .05       0
    5073     .08       0  5153.7     .05       0  5191.3     .08       0
  5331.6     .05       0    5477     .08       0  5645.6     .05       0
Bank Sta=4971.6,5036.6
XS Rating Curve= 0 ,0
Exp/Cntr=0.3,0.1

Type RM Length L Ch R = 1 ,60907   ,589,589,589
BEGIN DESCRIPTION:
WEST CANEY CREEK 70.0
END DESCRIPTION:
XS GIS Cut Line= 3
      3613887.99     10358188.77      3613015.92     10358088.94
      3612516.47     10358038.99
#Sta/Elev= 30
  4378.6  358.58  4595.9  356.99  4726.7  354.39  4777.1  354.48  4817.3  354.03
  4835.2  353.33  4897.9   352.9    4918  351.64  4923.9  350.34  4958.2  352.13
  4978.4  351.74  4995.3  346.53  4995.5  346.46  4998.3  345.96  5001.5  346.46
  5008.2  347.64  5013.2   347.6  5018.6  349.48  5028.7  351.32  5038.8  352.72
  5048.8  353.12  5191.7  355.61  5219.9  356.85  5260.8  357.08  5277.3  357.77
  5350.6  358.29  5377.8  358.96  5451.1   358.8  5684.4  359.82  5758.3  360.83
#Mann= 5 ,-1 , 0
  4378.6     .05       0  4835.2     .16       0  4995.3     .05       0
  4995.5     .03       0  5001.5     .05       0
Bank Sta=4978.4,5028.7
XS Rating Curve= 0 ,0
Exp/Cntr=0.3,0.1

Type RM Length L Ch R = 1 ,60318   ,891,891,891
BEGIN DESCRIPTION:
WEST CANEY CREEK 69.0
END DESCRIPTION:
XS GIS Cut Line= 3
      3613992.14     10357941.67       3613552.4     10357601.49
      3612605.69     10357551.23
#Sta/Elev= 30
  4171.7  363.28    4179  362.77  4185.3  360.81  4193.5  360.17  4199.8  358.47
  4214.3  357.55  4357.4   356.9  4563.7   352.6    4718  350.86  4812.8  349.98
  4923.4  348.75  4958.3  347.48  4968.3   348.8  4978.3   349.1  4988.3  347.62
  4995.3  343.72  4998.1  343.22  5001.3  343.72  5005.6  346.09  5010.6  344.29
  5022.1  346.96  5028.4  348.23  5048.4  350.66  5078.4  351.58  5088.5  352.62
  5108.5  353.43  5218.6  355.48  5327.4  355.04  5381.8  355.23  5675.7  355.53
#Mann= 9 ,-1 , 0
  4171.7     .05       0    4718     .16       0  4812.8     .05       0
  4923.4     .16       0  4995.3     .07       0  5001.3     .16       0
  5022.1     .05       0  5327.4      .1       0  5381.8     .05       0
Bank Sta=4988.3,5028.4
XS Rating Curve= 0 ,0
Exp/Cntr=0.3,0.1

Type RM Length L Ch R = 1 ,59427   ,1391,1391,1391
BEGIN DESCRIPTION:
WEST CANEY CREEK 68.0
END DESCRIPTION:
XS GIS Cut Line= 3
      3614341.04      10357433.7      3613946.71     10357156.84
      3612855.79      10357145.1
#Sta/Elev= 30
  4281.8  357.43  4427.1  356.55  4439.4  356.69  4448.1  358.03  4454.2  358.23
    4469   356.8  4498.6  356.95  4525.6  355.47    4591  353.59  4727.8  350.63
  4861.5  348.74  4918.2  349.09  4938.2  348.13  4968.2  347.75  4978.2  347.11
  4988.2   344.4  4995.2  341.43    4998  340.93  5001.2  341.43  5008.2  341.69
  5028.2  343.97  5068.2  345.05  5098.2  344.32  5129.3  345.18  5148.2  345.81
  5168.2  347.98  5208.2  349.76  5318.3  351.89  5678.3  353.96  5854.6  354.45
#Mann= 5 ,-1 , 0
  4281.8     .05       0  4861.5     .16       0  4995.2     .07       0
  5001.2     .16       0  5129.3     .05       0
Bank Sta=4988.2,5028.2
XS Rating Curve= 0 ,0
Exp/Cntr=0.3,0.1

Type RM Length L Ch R = 1 ,58036   ,1434,1434,1434
BEGIN DESCRIPTION:
WEST CANEY CREEK 67.0
END DESCRIPTION:
XS GIS Cut Line= 3
      3614433.35     10356670.26      3613929.94     10356351.43
      3612976.92     10356475.92
#Sta/Elev= 30
  4183.6  350.04  4394.1  348.96  4409.3  348.03    4567  345.72  4705.9  344.32
  4821.2  344.49  4868.1  343.55  4918.5  343.62  4938.7  342.78  4968.9  341.34
    4974  339.85  4979.1  340.23  4996.2  337.82  4998.9  337.32  5002.2  337.82
  5009.3  338.22  5029.4  343.03    5053  343.08  5079.8  345.81  5140.4  348.14
  5150.4  347.87  5205.8  349.28  5251.3  351.17  5346.7  350.46  5432.6  349.85
  5511.5  350.22  5553.8  351.73  5634.5  350.17    5695  351.27  5740.6  350.65
#Mann= 4 ,-1 , 0
  4183.6     .05       0  4996.2     .03       0  5002.2     .05       0
  5346.7     .12       0
Bank Sta=4938.7,5029.4
XS Rating Curve= 0 ,0
Exp/Cntr=0.3,0.1

Type RM Length L Ch R = 1 ,56602   ,1679,1679,1679
BEGIN DESCRIPTION:
WEST CANEY CREEK 66.0
END DESCRIPTION:
XS GIS Cut Line= 3
      3615775.63     10354740.63      3614533.99     10355537.63
      3613158.36      10355906.7
#Sta/Elev= 30
  3230.4  377.37  3292.6  374.92    3561  358.89  3589.9  357.27  3794.1  350.79
  4058.3  341.77  4094.6  337.63    4122  330.55  4124.7  330.05    4128  330.55
  4130.9  332.34  4152.1  331.67  4173.3  335.19  4236.6   336.3    4349  339.48
  4354.9  337.56  4391.2  341.99  4636.8  344.51  4792.2  343.03  4873.4  342.89
  4966.6  339.34  4977.2  337.69  4997.7  332.11  5039.1  337.65  5132.3  341.15
  5281.6  342.29  5484.3  346.44  5671.3  348.71  5807.9  348.43  6130.1  348.18
#Mann= 9 ,-1 , 0
  3230.4     .05       0    3561     .16       0  3589.9     .05       0
  3794.1     .16       0    4122     .07       0    4128     .16       0
  4236.6     .05       0  4792.2     .16       0  5807.9     .12       0
#XS Ineff= 2 , 0
         4638.64  344.96
Permanent Ineff=
       F       F
Bank Sta=4977.2,5039.1
XS Rating Curve= 0 ,0
Exp/Cntr=0.3,0.1

Type RM Length L Ch R = 1 ,54923   ,1176,1176,1176
BEGIN DESCRIPTION:
WEST CANEY CREEK 65.0
END DESCRIPTION:
XS GIS Cut Line= 3
      3615330.99     10353968.77        3614090.      10354572.6
      3613132.92     10355294.32
#Sta/Elev= 30
  3619.9  368.02  3704.3  364.11  3874.4  360.36  3957.9  354.19  4041.3  351.93
  4063.5  349.36  4098.7  349.17  4219.2   343.6  4608.4  333.53  4675.2  332.46
  4702.4  333.81  4735.6  332.07  4755.2  326.33  4757.9  325.83  4761.2  326.33
  4786.4  332.45  4825.8  330.94  4921.6  335.18  4956.5  332.14  4975.4  332.98
    4996  327.83  5005.2  327.04  5011.4  329.48    5037  331.72  5045.7  332.56
  5190.5  338.39  5361.2  342.43  6004.4  347.61  6062.1  346.84  6198.7  346.73
#Mann= 8 ,-1 , 0
  3619.9     .05       0  4702.4     .16       0  4755.2     .03       0
  4761.2     .16       0  4956.5     .05       0    5037     .16       0
  5045.7     .05       0  6062.1     .12       0
Bank Sta=4975.4,5045.7
XS Rating Curve= 0 ,0
Exp/Cntr=0.3,0.1

Type RM Length L Ch R = 1 ,53747   ,1065,1065,1065
BEGIN DESCRIPTION:
WEST CANEY CREEK 64.0
END DESCRIPTION:
XS GIS Cut Line= 3
      3614338.13     10353239.25      3613988.11     10353639.27
      3612892.09     10354791.66
#Sta/Elev= 30
  4114.5  364.47  4127.8  362.01  4191.4   358.3  4212.3  358.47  4383.1  350.53
  4389.7   351.2    4404  349.54  4439.1  349.94  4460.9  347.96  4510.3  346.44
  4602.3  345.38  4616.6  343.83  4701.6   341.9  4778.3  341.74  4941.9  336.99
    4956  335.22  4970.2  331.78  4977.4  328.68  4984.3  325.28  4995.5  321.86
  4998.2  321.36  5001.5  321.86  5026.8  328.35  5062.4  330.45  5111.6  330.76
  5287.6  330.76  5441.4   332.8  5776.7  338.38  5868.5  338.75  6236.4  344.16
#Mann= 7 ,-1 , 0
  4114.5     .05       0  4778.3     .16       0  4995.5     .07       0
  5001.5     .16       0  5111.6     .12       0  5287.6     .16       0
  5441.4     .05       0
Bank Sta=4977.4,5026.8
XS Rating Curve= 0 ,0
Exp/Cntr=0.3,0.1

Type RM Length L Ch R = 1 ,52682   ,1257,1257,1257
BEGIN DESCRIPTION:
WEST CANEY CREEK 63.0
END DESCRIPTION:
XS GIS Cut Line= 3
      3613418.19     10353020.68      3612864.44     10353859.69
      3612772.16     10354413.38
#Sta/Elev= 30
    4199  368.17  4456.4  352.38  4522.7  349.12  4705.4  336.66  4787.6   331.5
  4862.4  328.78    4905  327.69  4926.1  325.09  4962.2  327.24  4983.3  326.07
  4990.9  323.04  4995.3  320.31  4998.1  319.81  5001.3  320.31  5004.3  320.62
  5019.4  325.26  5026.9  326.13  5071.9  328.48  5112.7  329.89  5148.8  329.58
  5277.2   330.8  5427.8  333.22  5432.9  332.52    5480  332.94  5500.3  333.95
  5549.5  333.58  5554.5  334.19  5610.3  334.46  5615.4  333.93  5765.6   336.7
#Mann= 6 ,-1 , 0
    4199     .05       0  4705.4     .16       0  4862.4     .12       0
  4995.3     .07       0  5001.3     .12       0  5071.9     .05       0
Bank Sta=4983.3,5026.9
XS Rating Curve= 0 ,0
Exp/Cntr=0.3,0.1

Type RM Length L Ch R = 1 ,51425   ,1078,1078,1078
BEGIN DESCRIPTION:
WEST CANEY CREEK 61.0
END DESCRIPTION:
XS GIS Cut Line= 3
      3612461.73     10352534.14      3612050.83     10353484.61
      3611850.83     10353884.61
#Sta/Elev= 30
  4063.8  351.95  4204.8     347  4298.8   342.3  4366.1  340.65  4396.5  338.67
  4402.1  338.67  4432.6  336.11  4540.4  331.36  4550.1  331.78  4562.2  330.66
  4602.5  331.35    4608  330.47  4683.9  327.51  4783.3  324.53  4889.1  324.41
  4911.7  322.95  4929.7  324.29  4965.3  324.88  4973.2  323.75  4976.2  323.32
  4984.6  316.83  4987.4  316.33  4990.6  316.83  5005.7  319.91  5011.1  319.91
  5029.2  322.92  5094.9  326.71  5350.6  335.79  5517.9  337.91  5546.5  338.23
#Mann= 7 ,-1 , 0
  4063.8     .12       0  4396.5     .16       0  4402.1     .12       0
  4973.2     .16       0  4984.6     .07       0  4990.6     .16       0
  5517.9     .12       0
Bank Sta=4976.2,5029.2
XS Rating Curve= 0 ,0
Exp/Cntr=0.3,0.1

Type RM Length L Ch R = 1 ,50347   ,630,630,630
BEGIN DESCRIPTION:
WEST CANEY CREEK 60.0
END DESCRIPTION:
XS GIS Cut Line= 3
      3612042.12     10352491.63      3611744.08     10352789.67
      3611471.75     10353431.82
#Sta/Elev= 30
  4417.8  341.13  4460.2  338.77  4474.4  338.95  4488.5  337.22  4502.7  336.15
  4644.1  328.43  4672.4  327.16  4686.5  327.38  4728.9   324.4  4813.8  321.92
  4886.5  322.59  4971.8  322.04  4981.2  317.12  4986.6  317.45  4990.5  314.16
  4993.3  313.66  4996.5  314.16  5004.4  315.42  5010.3  317.87  5026.1  320.74
  5057.7  321.52  5063.1  322.85  5082.4  323.71  5115.9  323.47  5139.5  323.92
  5263.3  327.26  5374.3  331.47  5438.9  332.56  5468.9   333.6  5536.8  334.18
#Mann= 4 ,-1 , 0
  4417.8     .12       0  4990.5     .07       0  4996.5     .12       0
  5082.4     .16       0
Bank Sta=4971.8,5026.1
XS Rating Curve= 0 ,0
Exp/Cntr=0.3,0.1

Type RM Length L Ch R = 1 ,49717   ,876,876,876
BEGIN DESCRIPTION:
WEST CANEY CREEK 59.0
END DESCRIPTION:
XS GIS Cut Line= 3
      3611893.34     10352091.37      3611442.11     10352491.64
      3610792.12     10353141.63
#Sta/Elev= 30
  4411.6  337.62  4413.6  337.62  4525.9   335.1  4582.8  333.15  4646.4  332.37
  4880.6     322  4915.7  320.83  4944.1  320.65  4950.8  320.03  4972.5  320.13
  4979.2  319.25  4986.8  317.29  4993.5  312.01    4998  311.95  5000.7  311.45
    5004  311.95  5007.7  317.27  5011.4  319.72  5028.9  320.59  5043.1   320.6
  5085.5  319.15  5117.9   321.1  5170.3  321.19  5269.3  324.28  5382.5   325.1
  5396.6  325.77  5522.6   327.7  5651.2  329.64  5863.3   336.1    5934  337.61
#Mann= 6 ,-1 , 0
  4411.6     .16       0  4413.6     .12       0    4998     .07       0
    5004     .12       0  5117.9     .16       0  5522.6     .05       0
Bank Sta=4979.2,5011.4
XS Rating Curve= 0 ,0
Exp/Cntr=0.3,0.1

Type RM Length L Ch R = 1 ,48841   ,1287,1287,1287
BEGIN DESCRIPTION:
WEST CANEY CREEK 57.0
END DESCRIPTION:
XS GIS Cut Line= 3
      3611531.37     10351402.37      3610792.11     10352141.64
      3610442.11     10352691.64
#Sta/Elev= 30
  3933.3  334.53  4059.5  332.62    4201  328.18  4314.1  326.02  4342.4  324.92
  4483.8  322.57  4625.2  321.34  4653.5  320.45  4738.4  319.74  4794.9  319.87
  4908.1  318.91  4964.6  319.28  4975.2  318.03  4981.7  318.03  4986.4  316.41
  4998.6  315.21  5001.4  314.71  5004.6  315.21  5022.8  318.19    5038  319.06
  5109.2  318.16    5138  318.41  5153.2  320.35  5189.6  323.43    5320  328.92
  5392.8  331.05  5419.9  332.48  5535.9  334.29  5559.6  335.31  5630.7  336.63
#Mann= 3 ,-1 , 0
  3933.3     .05       0  4998.6     .03       0  5004.6     .05       0
Bank Sta=4964.6,5038
XS Rating Curve= 0 ,0
Exp/Cntr=0.3,0.1

Type RM Length L Ch R = 1 ,47554   ,805,805,805
BEGIN DESCRIPTION:
WEST CANEY CREEK 55.0
END DESCRIPTION:
XS GIS Cut Line= 3
      3611186.48     10351124.66      3610267.32      10351593.6
      3609509.21     10352183.09
#Sta/Elev= 30
  4140.2  351.34  4268.6  351.52  4481.9  331.03  4608.8  322.12  4880.6  316.51
  4908.5  317.11  4930.9  314.79  4953.3  317.22  4964.6  316.51  4975.5  315.28
  4987.1  308.91  4994.7  308.16  4997.5  307.66  5000.7  308.16  5019.9  311.63
  5025.6  314.44  5042.2  316.42  5064.4  318.05  5108.9  314.98  5114.5  317.06
  5131.1   315.1  5177.3  318.43  5253.4  321.68  5280.6  325.44  5309.5  323.68
  5487.8  323.79  5531.2  324.58    5552  327.77  5672.7  331.44  6132.4  335.67
#Mann= 5 ,-1 , 0
  4140.2     .05       0  4880.6     .16       0  4994.7     .07       0
  5000.7     .16       0  5177.3     .05       0
Bank Sta=4964.6,5042.2
XS Rating Curve= 0 ,0
Exp/Cntr=0.3,0.1

Type RM Length L Ch R = 1 ,46749   ,955,955,955
BEGIN DESCRIPTION:
WEST CANEY CREEK 54.0
END DESCRIPTION:
XS GIS Cut Line= 3
      3610842.54     10350520.57       3610045.5     10351267.27
      3609231.66     10351795.85
#Sta/Elev= 30
  4140.3  351.45  4148.5  350.89  4155.3  348.29  4176.8   346.1  4183.6  348.02
  4205.1  347.67  4399.3  331.77    4447  331.84  4473.8   328.8  4666.4  320.11
  4773.4  317.39  4806.9  316.46  4834.8  315.89  4848.9  313.42  4877.3  313.35
  4897.3  314.84  4940.8   315.3  4969.1  314.08  5001.3  306.49    5004  305.99
  5007.3  306.49  5011.6  311.33  5018.4     312  5025.8  315.21  5246.1   318.1
  5475.5  327.31  5671.8  332.79  5780.6  334.11  6083.1  334.53  6202.9   337.5
#Mann= 9 ,-1 , 0
  4140.3     .05       0  4399.3     .16       0    4447     .05       0
  4666.4     .16       0  4773.4     .05       0  4806.9     .12       0
  4897.3     .05       0  5001.3     .03       0  5007.3     .05       0
Bank Sta=4969.1,5025.8
XS Rating Curve= 0 ,0
Exp/Cntr=0.3,0.1

Type RM Length L Ch R = 1 ,45794   ,1089,1089,1089
BEGIN DESCRIPTION:
WEST CANEY CREEK 52.0
END DESCRIPTION:
XS GIS Cut Line= 3
      3610414.65     10350059.15      3609724.65      10350768.5
      3609174.67     10351218.49
#Sta/Elev= 30
  4212.8  348.02  4228.8  347.33  4315.3  340.93  4329.4     342  4350.8  339.54
  4371.9  340.48  4499.2   335.7  4640.7  325.02  4668.9   319.4  4690.3  321.79
    4768  316.33    4890  313.95  4897.1  313.86  4930.6  310.25    4966  312.79
  4980.2  311.09  4987.1  307.41  5005.5     305  5008.2   304.5  5011.5     305
  5015.4     308  5022.6  309.22  5029.6  312.98  5057.9  313.31  5291.9  315.83
  5547.5  324.42  5646.5  324.63  5668.8  327.38  5724.8   329.2    5913  331.73
#Mann= 7 ,-1 , 0
  4212.8     .16       0  4228.8     .12       0    4890     .05       0
  4897.1     .12       0  5005.5     .07       0  5011.5     .12       0
  5057.9     .05       0
Bank Sta=4966,5029.6
XS Rating Curve= 0 ,0
Exp/Cntr=0.3,0.1

Type RM Length L Ch R = 1 ,44705   ,660,660,660
BEGIN DESCRIPTION:
WEST CANEY CREEK 50.0
END DESCRIPTION:
XS GIS Cut Line= 3
      3610037.07     10349723.59       3609350.5     10350223.85
      3608887.75     10351065.87
#Sta/Elev= 30
  3938.8  344.78    4048  341.71  4251.2  331.88  4299.1  328.12  4420.4  318.38
  4520.8   313.5  4900.1  311.76    4962  312.12  4978.1  307.82  4983.8  308.63
  4996.9  302.24  4999.7  301.74  5002.9  302.24    5014  305.42  5021.7  309.72
  5043.5  308.18    5054  309.54  5097.3  311.45  5271.8  312.31  5293.6  313.73
  5322.1  322.25  5353.3  327.18  5505.8  326.75  5559.8   329.5  5646.9  330.72
  5668.7  331.54  5690.4  336.91  5698.6  338.05  5721.4  335.29  5749.1  335.17
#Mann= 9 ,-1 , 0
  3938.8     .05       0  4251.2     .16       0  4299.1     .05       0
  4900.1     .16       0  4996.9     .07       0  5002.9     .16       0
    5054     .12       0  5097.3     .16       0  5690.4     .05       0
Bank Sta=4983.8,5021.7
XS Rating Curve= 0 ,0
Exp/Cntr=0.3,0.1

Type RM Length L Ch R = 1 ,44045   ,712,712,712
BEGIN DESCRIPTION:
WEST CANEY CREEK 48.0
END DESCRIPTION:
XS GIS Cut Line= 3
      3609869.34     10349245.33      3609147.81     10349807.46
      3608417.87     10350503.84
#Sta/Elev= 30
  3897.3  338.42  4092.5  334.49    4306  323.35  4604.6  314.03  4967.5  308.93
  4979.6  304.72  4997.1  302.43  4999.8  302.08  5002.5  301.58  5005.8  302.08
  5016.9  308.15  5024.2  310.69  5073.2  309.85  5094.9  309.29  5109.1  305.55
    5116  307.28  5123.2  304.23  5130.1  308.13  5137.4   307.6  5144.3  310.05
  5179.5  309.62    5222  314.86  5236.1  313.67  5243.4  310.69  5321.1  310.04
  5335.2  310.34  5342.5  313.99  5349.4  314.43  5452.8  318.12  5820.8  337.29
#Mann= 7 ,-1 , 0
  3897.3     .05       0  4979.6     .16       0  4997.1     .12       0
  4999.8     .07       0  5005.8     .12       0  5073.2     .16       0
  5452.8     .05       0
#XS Ineff= 2 , 0
                         5223.01          314.92
Permanent Ineff=
       F       F
Bank Sta=4967.5,5016.9
XS Rating Curve= 0 ,0
Exp/Cntr=0.3,0.1

Type RM Length L Ch R = 1 ,43333   ,1095,1095,1095
BEGIN DESCRIPTION:
WEST CANEY CREEK 47.0
END DESCRIPTION:
XS GIS Cut Line= 3
      3609382.71     10348716.81      3608938.06     10349446.71
      3608175.88     10350108.38
#Sta/Elev= 30
  3794.4  351.26  3927.4  342.85  4285.9  315.57  4322.6  311.47  4365.3  311.49
  4386.6  309.41  4423.4  311.06  4438.8  307.53  4444.7  309.52  4454.3  306.58
  4460.2  307.78  4475.6  306.31  4481.5  308.27  4490.9  306.01  4510.9  309.97
  4591.8  311.64  4769.5  308.96  4954.5  309.44    4983  307.51  4989.6  303.46
  5000.9  302.78  5003.6  302.28  5006.9  302.78  5025.7  307.79  5060.7  308.88
  5089.3  308.04  5189.2  315.13  5196.1  315.35  5379.9  328.95  5658.4  336.91
#Mann= 9 ,-1 , 0
  3794.4     .12       0  3927.4     .16       0  4510.9     .05       0
  4769.5     .12       0  5000.9     .07       0  5006.9     .12       0
  5060.7     .05       0  5189.2     .16       0  5196.1     .05       0
Bank Sta=4983,5025.7
XS Rating Curve= 0 ,0
Exp/Cntr=0.3,0.1

Type RM Length L Ch R = 1 ,42238   ,871,871,871
BEGIN DESCRIPTION:
WEST CANEY CREEK 45.0
END DESCRIPTION:
XS GIS Cut Line= 3
      3608992.12     10348441.62      3608207.53     10349327.23
      3607957.86     10349526.97
#Sta/Elev= 30
  4213.6  341.04  4461.6  322.89  4532.7  315.07  4546.9  311.47  4553.6  308.69
  4574.5  306.08  4730.9  306.67  4766.1  308.21  4858.1  306.91    4894  307.63
  4908.3  307.12  4914.9  305.38  4929.2  304.37  4943.4  304.46  4950.1  306.79
  4957.6  305.99  4964.3  306.79  4978.5  305.17  4992.7  299.36  4997.3  298.64
    5000  298.14  5003.3  298.64  5014.5  305.49  5049.4  307.09  5184.3  308.16
  5439.8  323.58  5503.8  326.48    5539  327.34  5667.1  327.29  5716.5  325.93
#Mann= 4 ,-1 , 0
  4213.6     .12       0  4997.3     .07       0  5003.3     .12       0
  5049.4     .05       0
Bank Sta=4978.5,5014.5
XS Rating Curve= 0 ,0
Exp/Cntr=0.3,0.1

Type RM Length L Ch R = 1 ,41367   ,895,895,895
BEGIN DESCRIPTION:
WEST CANEY CREEK 44.0
END DESCRIPTION:
XS GIS Cut Line= 3
      3608896.11      10347986.9      3608057.83     10348715.84
      3606647.65     10348918.16
#Sta/Elev= 30
  4172.8  354.21  4323.1  345.93    4548  331.78  4575.7  325.89  4597.3   323.8
    4604  325.86  4632.4  321.96  4696.1  308.19  4781.5  305.01  4816.7  307.31
  4845.1   305.2  4965.7  305.56    4980  299.65  4986.6  301.42  4997.9  296.64
  5000.6  296.14  5003.9  296.64  5029.3  305.87  5155.8  305.88  5375.6  306.18
  5468.2  307.39  5612.7   308.5  5653.2   298.7  5683.5  308.11  5785.9  306.75
  5956.2  309.39  5986.5  311.82  6107.8  308.37  6410.8  315.31  6708.3     326
#Mann= 7 ,-1 , 0
  4172.8     .12       0  4323.1     .16       0  4997.9     .07       0
  5003.9     .16       0  5155.8     .05       0  5375.6     .16       0
  5468.2     .05       0
#XS Ineff= 2 , 0
                          5987.5          312.17
Permanent Ineff=
       F       F
Bank Sta=4965.7,5029.3
XS Rating Curve= 0 ,0
Exp/Cntr=0.3,0.1

Type RM Length L Ch R = 1 ,40472   ,1287,1287,1287
BEGIN DESCRIPTION:
WEST CANEY CREEK 43.0
END DESCRIPTION:
XS GIS Cut Line= 3
       3608392.7     10347642.94      3607942.11     10347941.64
      3606492.06     10348741.66
#Sta/Elev= 30
  4424.8     371  4497.5  370.52  4610.1  354.49  4648.1  348.14  4731.5   339.2
  4915.8  320.15  4942.8  308.25  4968.3  303.86  4988.2  295.46  4997.9   294.6
  5000.7   294.1  5003.9   294.6  5022.7  303.64  5060.5  305.29  5141.9  303.58
  5216.7  306.53  5239.3  304.35    5245  299.71  5266.8  302.17  5282.9  300.58
  5288.6  303.38  5332.1  306.31  5468.2  306.36  5583.5  306.54  5667.5  306.85
  5705.3  307.76    5799  308.76  6157.3   313.6    6445  327.86  6621.5  330.96
#Mann= 10 ,-1 , 0
  4424.8     .05       0  4610.1     .16       0  4731.5     .12       0
  4997.9     .07       0  5003.9     .12       0  5468.2     .05       0
  5583.5     .16       0  5667.5     .05       0  5705.3     .16       0
    5799     .05       0
Bank Sta=4968.3,5022.7
XS Rating Curve= 0 ,0
Exp/Cntr=0.3,0.1

Type RM Length L Ch R = 1 ,39185   ,972,972,972
BEGIN DESCRIPTION:
WEST CANEY CREEK 41.0
END DESCRIPTION:
XS GIS Cut Line= 3
      3608343.83      10347223.5       3607593.8     10347423.51
       3606192.1     10348141.65
#Sta/Elev= 30
  3928.4  359.51  4058.3   359.7  4173.4  355.25  4213.5  355.59  4368.8   341.6
    4599  316.78  4734.6  306.07    4906  301.09  4956.1  303.99  4978.3  301.15
  4987.4  297.46  4991.8  293.69  4994.6  293.19  4997.8  293.69  5009.9  293.91
    5017  299.24  5022.7  298.54  5032.4  304.32  5211.2  304.47  5239.1  301.52
  5245.9   298.9  5272.2  303.94  5366.7  308.03  5438.4  308.02  5694.1  307.89
  5810.7  310.97  5915.6  316.69  6139.4  329.94  6205.4     332  6279.6  332.71
#Mann= 9 ,-1 , 0
  3928.4     .05       0  4734.6     .12       0  4991.8     .07       0
  4997.8     .12       0  5272.2     .16       0  5438.4     .05       0
  5915.6     .16       0  6139.4     .12       0  6205.4     .16       0
Bank Sta=4978.3,5017
XS Rating Curve= 0 ,0
Exp/Cntr=0.3,0.1

Type RM Length L Ch R = 1 ,38213   ,1103,1103,1103
BEGIN DESCRIPTION:
WEST CANEY CREEK 39.0
END DESCRIPTION:
XS GIS Cut Line= 3
      3607906.13      10346359.3      3606471.45     10347524.26
      3606071.44     10347824.27
#Sta/Elev= 30
  3394.6  355.35  3485.5  353.36  3583.7  351.36  3669.9   344.3  3746.5  336.03
  3903.3  319.94  3981.6  314.01    4103   308.6  4315.7  307.07  4365.9  304.68
  4544.1  301.63  4695.4  302.37  4956.5  302.78  4970.8  301.74  4977.3  298.02
  4991.7  293.71  4995.1  291.04  4997.8  290.54  5001.1  291.04  5020.4  297.14
  5026.8  299.95    5062  301.94  5105.1  301.83  5148.1  305.03  5190.3  308.53
  5332.8  313.73  5364.4   317.3  5568.2  328.18  5724.7  329.79  5742.7  329.91
#Mann= 10 ,-1 , 0
  3394.6     .05       0  3485.5     .16       0  3669.9     .12       0
  3746.5     .16       0  4695.4     .12       0  4995.1     .07       0
  5001.1     .12       0  5148.1     .05       0  5364.4     .16       0
  5724.7     .12       0
Bank Sta=4977.3,5020.4
XS Rating Curve= 0 ,0
Exp/Cntr=0.3,0.1

Type RM Length L Ch R = 1 ,37110   ,1303,1303,1303
BEGIN DESCRIPTION:
WEST CANEY CREEK 38.0
END DESCRIPTION:
XS GIS Cut Line= 3
      3607243.34     10345990.16      3606040.08      10347165.8
      3605840.06     10347515.83
#Sta/Elev= 30
  3789.5  344.56  3897.5  348.73  3925.8   348.5  4022.9  337.08    4138  324.66
    4145  322.24  4159.1  320.59  4243.9  311.88  4328.9  305.36  4399.6  302.05
  4868.3  298.77    4910  299.93  4972.4  299.43  4986.5  296.05  4997.7   289.8
  5000.4   289.3  5003.7   289.8  5014.8  292.95  5028.9  300.76  5071.8  300.83
  5120.8  300.68  5340.1  309.88  5417.9  310.66  5446.1  309.64  5453.3  311.23
    5481  312.69  5518.4  310.59  5614.9  316.99  5868.2  324.03  5874.9  324.11
#Mann= 9 ,-1 , 0
  3789.5     .16       0  4022.9     .12       0  4243.9     .16       0
  4868.3     .12       0    4910     .16       0  4997.7     .07       0
  5003.7     .16       0  5071.8     .05       0  5868.2     .16       0
Bank Sta=4972.4,5028.9
XS Rating Curve= 0 ,0
Exp/Cntr=0.3,0.1

Type RM Length L Ch R = 1 ,35807   ,774,774,774
BEGIN DESCRIPTION:
WEST CANEY CREEK 37.0
END DESCRIPTION:
XS GIS Cut Line= 3
      3606966.52     10345730.05      3605951.33     10346342.52
      3605665.29     10347111.83
#Sta/Elev= 30
  4096.8  345.16  4151.4   343.7  4209.6  337.79  4253.8  330.81  4267.9  330.58
  4399.9  316.51    4523  306.81  4602.5   302.7  4641.1  303.77  4712.4  299.82
  4759.3  298.97  4960.8  299.05  4982.2  298.17  4989.6   293.7  4997.7  288.28
  5009.9  287.04  5012.7  286.54  5015.9  287.04  5019.1  290.25  5034.6  294.67
  5040.4  293.82  5047.9   298.3  5061.8  299.34  5531.7  299.47  5663.9  299.91
    5871  304.96    5975  309.27  6012.1  313.04  6037.1  312.99  6103.2  317.54
#Mann= 8 ,-1 , 0
  4096.8     .16       0    4523     .07       0  4602.5      .1       0
  4641.1     .07       0  4759.3     .12       0  5009.9     .07       0
  5015.9     .12       0  5531.7     .16       0
Bank Sta=4989.6,5034.6
XS Rating Curve= 0 ,0
Exp/Cntr=0.3,0.1

Type RM Length L Ch R = 1 ,35033   ,1239,1239,1239
BEGIN DESCRIPTION:
WEST CANEY CREEK 36.0
END DESCRIPTION:
XS GIS Cut Line= 3
      3606692.08     10345341.65      3605308.18       10345797.
      3604316.25      10346258.2
#Sta/Elev= 30
  4140.5  330.02  4283.5  312.81  4507.2  301.43  4562.8  301.32  4951.1  296.77
  4972.1  293.72  5000.7  286.16  5003.5  285.66  5006.7  286.16  5025.2  293.21
  5035.3   297.1    5057  297.89  5077.4  295.68  5083.5   290.6  5088.8  293.68
  5098.5     289  5115.3  292.04  5120.6  289.22  5152.3  290.46  5172.2  287.41
  5203.7  297.48  5242.4   297.5  5265.1  293.66    5306  297.79  5702.5  298.25
  5802.2  297.64  5906.1  298.55  5951.9  307.43  5974.8  308.12  6691.3  318.99
#Mann= 8 ,-1 , 0
  4140.5     .12       0  4507.2     .05       0  4562.8     .12       0
  5000.7     .07       0  5006.7     .12       0  5265.1     .05       0
  5702.5     .16       0  5802.2     .05       0
Bank Sta=4972.1,5025.2
XS Rating Curve= 0 ,0
Exp/Cntr=0.3,0.1

Type RM Length L Ch R = 1 ,33794   ,644,644,644
BEGIN DESCRIPTION:
WEST CANEY CREEK 35.0
END DESCRIPTION:
XS GIS Cut Line= 3
      3606345.67     10344186.35      3605473.12      10344723.3
      3604130.75     10345923.04
#Sta/Elev= 30
    3622  332.45  3648.5  332.99  3825.1  332.72  3852.1  330.94  4028.3  314.45
  4062.8  312.51  4181.7   305.4  4300.6  303.08  4380.6  301.57  4411.3  300.84
  4575.1  297.67  4585.5   297.6  4696.6   295.6  4861.7  295.81  4922.2  295.48
  4950.7  289.47  4979.1  289.46    4997  282.93  4999.7  282.43    5003  282.93
  5014.2  289.73  5028.4  294.96  5056.5  295.48  5120.4  294.15  5389.6  303.66
  5552.6  302.27    5744  308.29  5871.1  307.15  6274.8  316.06  6446.9  316.14
#Mann= 17 ,-1 , 0
    3622     .16       0  3648.5     .05       0  3825.1     .16       0
  3852.1     .12       0  4028.3     .16       0  4062.8     .05       0
  4181.7     .16       0  4300.6     .05       0  4380.6     .16       0
  4411.3     .05       0  4575.1     .16       0  4585.5     .05       0
  4696.6     .16       0  4861.7     .12       0    4997     .07       0
    5003     .12       0  5056.5     .05       0
Bank Sta=4979.1,5014.2
XS Rating Curve= 0 ,0
Exp/Cntr=0.3,0.1

Type RM Length L Ch R = 1 ,33150   ,2175,2175,2175
BEGIN DESCRIPTION:
WEST CANEY CREEK 33.0
END DESCRIPTION:
XS GIS Cut Line= 3
       3605716.4     10343632.66      3604759.99     10344773.64
      3604156.53     10345611.79
#Sta/Elev= 30
  3785.8  330.27  3939.2  325.24  4127.6  308.87  4244.1  302.74  4412.3  298.04
  4611.6  295.46  4616.2  295.47  4772.9  294.41  4885.7  294.68  4923.6  291.99
  4952.3  293.46  4973.1  292.36  4980.9  289.34  4987.4  284.18  4998.7  281.53
  5001.5  281.03  5004.7  281.53  5009.5  281.71    5016  288.65  5023.8  291.13
  5030.3  293.74  5044.6  295.18  5088.4   293.9  5165.6  294.53  5207.3  292.15
  5229.4  293.91    5436   294.1  5874.2  309.43  6016.6   308.3  6307.4  312.21
#Mann= 11 ,-1 , 0
  3785.8     .16       0  3939.2     .12       0  4127.6     .16       0
  4244.1     .05       0  4611.6     .16       0  4616.2     .05       0
  4772.9     .16       0  4885.7     .12       0  4998.7     .07       0
  5004.7     .12       0  5088.4     .05       0
Bank Sta=4973.1,5023.8
XS Rating Curve= 0 ,0
Exp/Cntr=0.3,0.1

Type RM Length L Ch R = 1 ,30975   ,2184,2184,2184
BEGIN DESCRIPTION:
WEST CANEY CREEK 32.0
END DESCRIPTION:
XS GIS Cut Line= 3
      3603879.07     10342953.03      3603864.02     10345088.72
      3603714.23     10345837.65
#Sta/Elev= 30
  3011.5  328.57  3060.1  327.45  3160.1  321.72  3320.1  308.92  3610.1  294.77
  4040.1  290.77  4110.1  291.79  4160.1  289.34  4270.1  292.44  4409.3  291.17
  4510.1  290.06  4610.1   291.2  4790.2  290.24  4940.2  292.51  4950.2  292.37
  4960.2  288.89  4997.2  279.54  4999.9  279.04  5003.2  279.54  5010.2  279.65
  5040.2  290.54  5050.2  291.79  5070.2  292.08  5120.2  304.73  5146.2  307.96
  5286.2  307.04  5527.5  308.72  5643.1  311.02    5791  315.63    5911  316.61
#Mann= 5 ,-1 , 0
  3011.5     .05       0  4409.3     .16       0  4997.2     .07       0
  5003.2     .16       0  5286.2     .05       0
Bank Sta=4960.2,5040.2
XS Rating Curve= 0 ,0
Exp/Cntr=0.3,0.1

Type RM Length L Ch R = 1 ,28791   ,733,733,733
BEGIN DESCRIPTION:
WEST CANEY CREEK 31.0
END DESCRIPTION:
XS GIS Cut Line= 3
      3603484.75     10343095.72      3603149.17     10344085.69
      3603341.92     10345778.56
#Sta/Elev= 30
  4355.5  341.17  4446.6  341.26  4504.1  336.86  4566.9  329.36  4593.1  323.53
  4655.9  314.96  4881.1  293.45  4955.8  282.36    4970  283.36  4975.3  279.99
  4984.7  281.82  5013.4  274.67  5016.2  274.17  5019.4  274.67    5027  275.24
  5038.1  283.07  5048.1  287.67  5058.6  288.89  5069.5  288.72  5095.7  282.72
  5100.9  284.98  5143.1  288.68  5227.6  290.71  6117.5  289.23  6212.6  290.95
  6302.5  303.79  6440.8  300.61  6544.1  303.23  6725.3   302.5  7104.6  311.65
#Mann= 6 ,-1 , 0
  4355.5     .05       0  4955.8     .16       0  5013.4     .07       0
  5019.4     .16       0  6117.5     .16       0  6212.6     .05       0
Bank Sta=4984.7,5038.1
XS Rating Curve= 0 ,0
Exp/Cntr=0.3,0.1

Type RM Length L Ch R = 1 ,28058   ,965,965,965
BEGIN DESCRIPTION:
WEST CANEY CREEK 30.0
END DESCRIPTION:
XS GIS Cut Line= 3
      3602821.98     10342894.31      3602528.33     10343951.45
      3602083.87     10345687.38
#Sta/Elev= 30
  4304.9  343.01  4343.7  339.95  4447.4  327.17  4512.4   322.1  4546.7  317.78
    4694  306.43  4807.2  295.79  4904.1  290.41  4935.2  286.62  4959.7  286.13
  4966.4  284.34  4976.7  282.61  4987.1  278.73    4991  275.49  4993.7  274.99
    4997  275.49  5007.9  278.15  5018.3  283.43  5028.2  287.35  5072.9  288.46
    5122  285.66  5194.7  289.25  5433.2  287.21  5932.5  288.03  6269.4  291.75
  6294.6  288.83  6310.7  291.44  6486.1  294.74  6795.8   306.3    7194  313.94
#Mann= 3 ,-1 , 0
  4304.9     .05       0    4991     .03       0    4997     .05       0
Bank Sta=4966.4,5018.3
XS Rating Curve= 0 ,0
Exp/Cntr=0.3,0.1

Type RM Length L Ch R = 1 ,27093   ,877,877,877
BEGIN DESCRIPTION:
WEST CANEY CREEK 29.0
END DESCRIPTION:
XS GIS Cut Line= 3
      3602251.47     10342709.78      3601601.75     10343742.09
      3600842.09     10344691.66
#Sta/Elev= 30
  4179.9  333.95  4224.5  333.15  4412.9  321.07    4586  307.63    4659  304.41
  4820.2   292.6  4899.2  284.57  4962.8  283.52  4972.2  280.89  4985.6  273.18
  4990.4  272.09  4993.2  271.59  4996.4  272.09  5008.7  277.94  5014.6  282.83
  5035.8  285.56  5080.1  283.41  5139.2  286.47  5519.9  285.64  5612.8   282.9
  5683.2  285.87  5790.5  285.18  5825.7  282.03  5875.3  280.82  5883.3  282.18
  5932.9  282.18  5982.6  287.66  6288.3  296.41  6509.2   306.7  6615.7  308.25
#Mann= 3 ,-1 , 0
  4179.9     .05       0  4990.4     .03       0  4996.4     .05       0
Bank Sta=4962.8,5014.6
XS Rating Curve= 0 ,0
Exp/Cntr=0.3,0.1

Type RM Length L Ch R = 1 ,26216   ,1525,1525,1525
BEGIN DESCRIPTION:
WEST CANEY CREEK 28.0
END DESCRIPTION:
XS GIS Cut Line= 3
      3601840.35     10342441.33      3600832.72     10343504.95
      3600204.67     10344336.99
#Sta/Elev= 30
  3776.4  314.09  3804.7  312.64  3837.6  311.96  3943.2  307.07  3966.7  306.54
  4220.9  293.34  4348.3  289.63  4859.3  283.67  4949.5  284.68  4956.7  275.94
  4982.1  270.35  4984.8  269.85  4988.1  270.35  5006.1  271.85  5013.4  280.01
  5020.3  279.76  5027.5  283.79  5184.3  284.15  5411.7  282.67  5438.8  275.36
  5453.3  278.07  5461.6  276.43  5467.9  279.07  5482.5  276.23  5488.7  281.04
  5503.3  282.96  5811.3  284.99  5932.1   289.2  6125.6  301.95    6284  308.57
#Mann= 9 ,-1 , 0
  3776.4     .16       0  3804.7     .12       0  3837.6     .16       0
  3943.2     .12       0  3966.7     .05       0  4859.3     .12       0
  4982.1     .07       0  4988.1     .12       0  5184.3     .05       0
Bank Sta=4949.5,5027.5
XS Rating Curve= 0 ,0
Exp/Cntr=0.3,0.1

Type RM Length L Ch R = 1 ,24691   ,765,765,765
BEGIN DESCRIPTION:
WEST CANEY CREEK 26.0
END DESCRIPTION:
XS GIS Cut Line= 3
      3600942.08     10341491.67      3599606.18     10343402.06
      3599456.65      10343800.8
#Sta/Elev= 30
    3269  332.02  3368.8  328.67  3556.3  314.25    3613  312.55  3678.4  308.72
  3785.7  305.86  3886.8  299.42  4044.7  292.12  4151.9  289.11  4181.6  286.84
  4553.9  282.98  4726.6  282.88  4855.3  280.88  4941.1  282.98  4964.7  281.29
  4977.3  272.61  4988.7  268.29  4991.4  267.79  4994.7  268.29  5006.5  271.29
  5013.9  277.34  5021.3  279.95  5027.4   282.5  5164.4  282.76  5229.8  279.01
  5316.1  288.18  5473.9  294.27  5620.8  297.77  5802.6   298.2    6026  303.02
#Mann= 3 ,-1 , 0
    3269     .05       0  4988.7     .03       0  4994.7     .05       0
Bank Sta=4964.7,5021.3
XS Rating Curve= 0 ,0
Exp/Cntr=0.3,0.1

Type RM Length L Ch R = 1 ,23926   ,243,243,243
BEGIN DESCRIPTION:
WEST CANEY CREEK 25.0
END DESCRIPTION:
XS GIS Cut Line= 4
      3600212.76     10341979.88      3599389.01     10342758.21
      3599057.59     10342896.05      3598706.57     10343333.74
#Sta/Elev= 30
  3866.7  288.57  4017.1  285.23  4462.5   281.2  4872.7   281.5  4950.8  281.07
  4979.1  276.03  4995.9  269.27  4998.6  268.77  5001.9  269.27  5022.8  273.06
  5029.1  276.56  5046.7  282.12  5094.1  280.71  5115.8  272.67  5123.7  271.55
  5137.4  273.95  5147.5  278.41    5187  279.94  5213.3  283.05  5259.2  284.15
  5306.9  283.03  5424.4  284.89  5428.6   285.3  5502.1  283.69  5545.3  284.37
  5572.6  287.04  5609.4  286.29  5790.5  299.33  5915.7  306.84    5920  306.94
#Mann= 9 ,-1 , 0
  3866.7     .05       0  4872.7     .16       0  4995.9     .07       0
  5001.9     .16       0    5187     .05       0  5424.4     .16       0
  5428.6     .05       0  5790.5     .16       0  5915.7     .05       0
Bank Sta=4979.1,5029.1
XS Rating Curve= 0 ,0
Exp/Cntr=0.3,0.1

Type RM Length L Ch R = 1 ,23683   ,558,558,558
BEGIN DESCRIPTION:
WEST CANEY CREEK 24.0
END DESCRIPTION:
XS GIS Cut Line= 4
      3599826.85     10341820.47      3599553.27     10342327.11
      3599292.11     10342541.64      3598642.07     10343141.67
#Sta/Elev= 30
  4089.4  288.15  4545.3  280.59  4790.1  279.68    4852  280.23  4890.8  280.11
  4925.5  281.29  4957.3  279.43  4967.3  278.43  4975.2  274.33  4981.6  276.16
  4989.5   270.2    4996  269.12  4996.9  267.47  4999.7  266.97  5002.9  267.47
  5017.1  268.93  5031.2   274.9  5038.6  275.79  5045.4  279.93  5052.8   279.5
  5059.6  281.13  5105.7  280.95    5173  279.73  5215.5  281.69  5399.2   282.9
  5498.5  285.42  5611.9  286.56  5654.4  287.98  5732.1  292.49  5887.8  304.25
#Mann= 7 ,-1 , 0
  4089.4     .05       0    4852     .16       0  4890.8     .05       0
  4957.3     .16       0  4996.9     .07       0  5002.9     .16       0
  5105.7     .05       0
Bank Sta=4981.6,5038.6
XS Rating Curve= 0 ,0
Exp/Cntr=0.3,0.1

Type RM Length L Ch R = 1 ,23125   ,1019,1019,1019
BEGIN DESCRIPTION:
WEST CANEY CREEK 23.0
END DESCRIPTION:
XS GIS Cut Line= 3
      3599665.22     10341191.42      3598942.11     10342241.64
      3598354.84     10343057.21
#Sta/Elev= 30
  3751.5  313.92  4120.3  292.86  4257.6  286.83  4630.9  276.94  4741.4  279.65
  4881.8  278.88  4932.6  280.45  4962.4   280.2  4968.4  279.13  4977.2  277.74
  4983.3  272.61  5001.3  266.14    5004  265.64  5007.3  266.14  5019.2  268.37
  5023.6  270.86  5029.7  270.86  5035.1  272.42  5040.1  274.81  5048.7  274.06
  5054.8  279.68  5063.4  280.76  5155.5   279.5  5392.3  280.29  5470.2  281.99
  5670.9  282.88  5886.9  295.12  5972.8  298.68  5993.7  297.66  6031.6  298.87
#Mann= 5 ,-1 , 0
  3751.5     .05       0  4741.4     .16       0  5001.3     .07       0
  5007.3     .16       0  5035.1     .05       0
Bank Sta=4968.4,5054.8
XS Rating Curve= 0 ,0
Exp/Cntr=0.3,0.1

Type RM Length L Ch R = 1 ,22106   ,798,798,798
BEGIN DESCRIPTION:
WEST CANEY CREEK 21.0
END DESCRIPTION:
XS GIS Cut Line= 3
      3599092.11     10340841.64      3598451.36     10341442.34
      3597938.08      10343247.7
#Sta/Elev= 30
  3851.8  315.45  3915.5  310.16  4031.3  304.64  4066.6  303.32  4396.7  285.86
  4481.7  283.02  4864.5  276.77  4958.1   278.7  4964.2  276.46  4969.4  277.81
  4980.3  269.76  4989.3  265.36  5000.2  264.08    5003  263.58  5006.2  264.08
  5020.5  267.69  5037.1  276.54  5042.3   275.9  5051.6  277.79  5200.5  277.65
  5261.2  278.61    5665  277.53  5997.7  281.29  6153.7  284.61    6268  291.12
  6382.4  294.75  6403.2  292.57  6423.2  292.39  6467.5  296.77    6607   300.5
#Mann= 7 ,-1 , 0
  3851.8     .05       0  4031.3     .16       0  4066.6     .05       0
  4980.3     .16       0  5000.2     .07       0  5006.2     .16       0
  5200.5     .05       0
Bank Sta=4969.4,5051.6
XS Rating Curve= 0 ,0
Exp/Cntr=0.3,0.1

Type RM Length L Ch R = 1 ,21308   ,631,631,631
BEGIN DESCRIPTION:
WEST CANEY CREEK 20.0
END DESCRIPTION:
XS GIS Cut Line= 3
      3598692.08     10340591.66      3597972.52     10341095.92
      3597382.24     10343431.01
#Sta/Elev= 30
  3785.9   308.3  4131.2  289.98  4281.4  285.09  4323.3   282.6  4495.9  278.92
  4670.5  276.67  4856.1  277.05  4891.4  274.78  4907.7  276.88  4938.6  277.66
  4968.4   275.5  4990.2     266    5009  262.65  5011.5  262.37  5014.3  261.87
  5017.5  262.37  5021.2  265.36  5041.8  274.99  5055.6   277.7  5109.3  276.89
  5173.5  276.09    5279  278.58  5501.8  276.39  5747.9  276.13  6124.8  278.21
  6372.4  281.43  6563.4  285.32  6914.5  295.39  6973.7  296.45  7073.1  300.94
#Mann= 7 ,-1 , 0
  3785.9     .16       0  4131.2     .05       0    5009     .12       0
  5011.5     .03       0  5017.5     .12       0  5109.3     .05       0
  6914.5     .12       0
Bank Sta=4968.4,5041.8
XS Rating Curve= 0 ,0
Exp/Cntr=0.3,0.1

Type RM Length L Ch R = 1 ,20677   ,1740,1740,1740
BEGIN DESCRIPTION:
WEST CANEY CREEK 19.0
END DESCRIPTION:
XS GIS Cut Line= 3
      3598345.77     10339984.83      3597477.73     10340783.42
      3596974.26     10343396.25
#Sta/Elev= 30
  3294.6  315.22  3500.3  304.15  4080.5  278.96  4420.2  275.03  4741.9   277.3
  4961.1  275.95  4971.3  273.97  4976.3  271.36  4991.7  262.83  4998.3  262.18
  5001.1  261.68  5004.3  262.18  5032.4  274.79  5042.6  276.11  5091.9  276.02
  5144.4  276.44  5225.9  271.44  5276.8  276.35  5516.6  275.74  5758.7  276.18
  6064.5  279.24  6346.1  285.02  6593.6  287.74  6682.2  291.23  6795.2  292.71
    6853  293.71  6897.8  292.51  7024.1  294.31  7072.1  295.19    7135  297.08
#Mann= 12 ,-1 , 0
  3294.6     .05       0  4976.3     .16       0  4998.3     .07       0
  5004.3     .16       0  5091.9     .05       0  5516.6     .16       0
  5758.7     .05       0  6346.1     .12       0  6795.2     .05       0
  6897.8     .16       0  7024.1     .05       0  7072.1     .16       0
Bank Sta=4961.1,5042.6
XS Rating Curve= 0 ,0
Exp/Cntr=0.3,0.1
