--- PLUMMERS CREEK.prj (project) ---

Proj Title=PLUMMERS CREEK Base Level Engineering
Current Plan=p01
Default Exp/Contr=0.3,0.1
English Units
Geom File=g01
Flow File=f01
Plan File=p01
Y Axis Title=Elevation
X Axis Title(PF)=Main Channel Distance
X Axis Title(XS)=Station
BEGIN DESCRIPTION:
PLUMMERS CREEK
END DESCRIPTION:
DSS Export Rating Curves= 0
DSS Export Rating Curve Sorted= 0
DSS Export Volume Flow Curves= 0
DXF OffsetX= 0
DXF OffsetY= 0
DXF ScaleX= 1
DXF ScaleY= 10

--- PLUMMERS CREEK.p01 (plan) ---

Plan Title=Multiple Run
Short Identifier=Multiple
Geom File=g01
Flow File=f01
Subcritical Flow
K Sum by GR= 0
Std Step Tol= 0.01
Critical Tol= 0.01
Num of Std Step Trials= 20
Max Error Tol= 0.3
Flow Tol Ratio= 0.001
Split Flow NTrial= 30
Split Flow Tol= 0.02
Split Flow Ratio= 0.02
Log Output Level= 0
Friction Slope Method= 1
Unsteady Friction Slope Method= 2
Unsteady Bridges Friction Slope Method= 1
Parabolic Critical Depth
Global Vel Dist=  1 , 1 , 1
Global Log Level= 0
CheckData=True
Encroach Param= -1, 0, 0, 0
BEGIN DESCRIPTION:
Multiple Run
END DESCRIPTION:

--- PLUMMERS CREEK.f01 (steady flow) ---

Flow Title=Multiple
Program Version=4.10
Number of Profiles= 7
Profile Names=10-year,25-year,50-year,1pct_min,100-year,1pct_plu,500-year
River Rch & RM=PLUMMERS CREEK,Reach-1         ,100345
     485     605     691     574     776    1049     977
River Rch & RM=PLUMMERS CREEK,Reach-1         ,91942
     653     825     953     798    1079    1459    1382
River Rch & RM=PLUMMERS CREEK,Reach-1         ,88818
     784    1000    1160     976    1321    1786    1708
River Rch & RM=PLUMMERS CREEK,Reach-1         ,82137
     917    1176    1371    1159    1567    2119    2043
River Rch & RM=PLUMMERS CREEK,Reach-1         ,79423
    1151    1490    1747    1484    2007    2714    2644
River Rch & RM=PLUMMERS CREEK,Reach-1         ,71532
    1247    1619    1902    1618    2188    2960    2893
River Rch & RM=PLUMMERS CREEK,Reach-1         ,64373
    1536    2010    2374    2030    2745    3713    3665
River Rch & RM=PLUMMERS CREEK,Reach-1         ,59903
    1798    2363    2799    2399    3244    4387    4350
River Rch & RM=PLUMMERS CREEK,Reach-1         ,52133
    1914    2520    2989    2564    3468    4690    4660
River Rch & RM=PLUMMERS CREEK,Reach-1         ,42357
    2273    3012    3586    3089    4177    5649    5656
River Rch & RM=PLUMMERS CREEK,Reach-1         ,39215
    2989    3988    4773    4128    5582    7550    7622
River Rch & RM=PLUMMERS CREEK,Reach-1         ,33955
    3073    4096    4899    4234    5726    7743    7805
River Rch & RM=PLUMMERS CREEK,Reach-1         ,26365
    3149    4187    4999    4312    5831    7886    7918
River Rch & RM=PLUMMERS CREEK,Reach-1         ,15003
    3511    4677    5592    4829    6531    8832    8886
Boundary for River Rch & Prof#=PLUMMERS CREEK,Reach-1         , 1
Up Type= 0
Dn Type= 3
Dn Slope=0.002
Boundary for River Rch & Prof#=PLUMMERS CREEK,Reach-1         , 2
Up Type= 0
Dn Type= 3
Dn Slope=0.002
Boundary for River Rch & Prof#=PLUMMERS CREEK,Reach-1         , 3
Up Type= 0
Dn Type= 3
Dn Slope=0.002
Boundary for River Rch & Prof#=PLUMMERS CREEK,Reach-1         , 4
Up Type= 0
Dn Type= 3
Dn Slope=0.002
Boundary for River Rch & Prof#=PLUMMERS CREEK,Reach-1         , 5
Up Type= 0
Dn Type= 3
Dn Slope=0.002
Boundary for River Rch & Prof#=PLUMMERS CREEK,Reach-1         , 6
Up Type= 0
Dn Type= 3
Dn Slope=0.002
Boundary for River Rch & Prof#=PLUMMERS CREEK,Reach-1         , 7
Up Type= 0
Dn Type= 3
Dn Slope=0.002
DSS Import GetInterval= 0
DSS Import GetPeak= 0
DSS Import FillOption= 0

--- PLUMMERS CREEK.g01 (geometry) ---

Geom Title=Existing Conditions
Program Version=4.10

River Reach=PLUMMERS CREEK  ,Reach-1
Reach XY= 30
      3484082.11     10604721.64      3486210.05     10599940.37
      3486269.21     10595018.41      3488037.99     10591854.65
      3487891.18     10590190.51      3491076.96     10587704.09
      3490304.23     10584952.77      3492808.55     10583694.19
      3492863.54     10582934.93      3496016.53     10582693.38
      3495995.51     10580722.97      3496939.23     10580241.22
      3495952.54     10575878.57      3496440.24     10574886.79
       3495492.2     10572722.03      3494276.34     10571998.19
      3493793.46     10570015.71      3493824.51     10568367.43
      3494712.11     10567771.64       3494603.1     10563409.14
      3492852.01     10557570.67      3492975.61     10555823.08
      3494327.93     10553759.11      3495858.52     10553115.25
      3497548.81     10550800.02      3497232.78     10549391.82
      3499119.39     10546800.19      3498647.54     10545889.11
      3499722.16     10545566.69      3498562.11     10542751.64

Type RM Length L Ch R = 1 ,100345  ,1083,1083,1083
BEGIN DESCRIPTION:
PLUMMERS CREEK 107.0
END DESCRIPTION:
XS GIS Cut Line= 5
      3485443.42     10605166.44        3484558.     10604437.28
      3483818.42     10604713.32      3482891.34     10604588.32
      3482891.34     10604577.93
#Sta/Elev= 30
  3353.3  543.49  3591.8  537.13  3805.6  533.23  4174.3  528.77  4701.4  527.11
  4762.8  525.65  4794.8  525.91  4811.9  528.68  4817.3  526.74  4836.9  529.22
  4842.3   527.9  4848.2  529.22  4867.2  528.39  4872.6   529.4  4897.5  525.73
  4902.9  527.41  4922.5  524.96  4927.9  526.15  4976.3  525.31  5007.9   520.8
    5019  524.31 5027.22  525.29    5051  526.42  5068.7  525.33  5074.1  526.49
    5099  524.86  5558.5  530.07  5901.5   539.2  6165.9  544.22  6235.6  544.29
#Mann= 3 , 0 , 0
  3353.3     .05       0  4976.3    .035       0 5027.22     .05       0
#XS Ineff= 2 , 0
       0  4976.3  525.31 5027.22       0  525.29
Permanent Ineff=
       T       T
Bank Sta=4976.3,5027.22
XS Rating Curve= 0 ,0
Exp/Cntr=0.3,0.1

Type RM Length L Ch R = 1 ,99262   ,84,84,84
BEGIN DESCRIPTION:
PLUMMERS CREEK 106.0
END DESCRIPTION:
XS GIS Cut Line= 4
      3485698.62     10604942.48      3484526.75     10604036.23
      3484094.46     10603708.11      3483719.43     10603442.46
#Sta/Elev= 30
  3308.1  548.61  3328.3  546.62  3334.6  543.93  3384.4  540.57  3606.3  538.33
  3755.7   534.8    3791  534.48    3820  536.53  3861.7  532.87  3919.6  531.59
  4289.7  527.79  4496.5  528.35  4531.8   526.7  4567.8  529.39  4596.1  524.43
  4631.4  526.52  4917.9  521.34  4974.1  523.01 4978.05  522.54  5002.9  517.82
  5009.4  520.93  5017.7  520.15  5038.5  522.68  5302.2  524.38  5474.6  527.54
  5511.8  529.85  5567.9  536.37  5611.2  531.17  5646.9  530.79  5791.8   536.5
#Mann= 5 ,-1 , 0
  3308.1     .05       0  4974.1    .035       0  5038.5     .05       0
  5302.2     .12       0  5511.8     .05       0
Bank Sta=4978.05,5038.5
XS Rating Curve= 0 ,0
Exp/Cntr=0.3,0.1

Type RM Length L Ch R = 1 ,99178   ,213,213,213
BEGIN DESCRIPTION:
PLUMMERS CREEK 105.2
END DESCRIPTION:
XS GIS Cut Line= 4
      3485745.49     10604890.39      3484636.13     10603937.28
      3484302.79     10603807.07      3483724.68     10603374.78
#Sta/Elev= 30
  3304.1  541.69  3617.6  537.57  3730.6  533.94  4043.3  530.29  4362.7  527.65
  4468.7  528.84  4504.2   526.6  4539.4  529.17  4582.2  525.99    4603  526.87
  4639.2   525.2    4738  525.21  4921.3  521.24  4953.5  521.52    4975   525.3
  4984.3  523.54 4986.69  522.44  4996.2   518.5  5014.2     521    5044  522.43
  5050.1  522.71    5093  524.31    5352  524.63  5493.2   526.9  5578.6  535.97
  5607.8  531.26  5621.3  530.99  5728.7  531.33  5787.1  536.56  5846.4  537.36
#Mann= 5 ,-1 , 0
  3304.1     .05       0  4984.3    .035       0  5050.1     .05       0
    5352     .12       0  5621.3     .05       0
#XS Ineff= 2 , 0
       0 4986.69  522.44    5044       0  522.43
Permanent Ineff=
       T       T
Bank Sta=4986.69,5044
XS Rating Curve= 0 ,0
Exp/Cntr=0.3,0.1

Type RM Length L Ch R = 1 ,98965   ,88,88,88
BEGIN DESCRIPTION:
PLUMMERS CREEK 105.1
END DESCRIPTION:
XS GIS Cut Line= 4
      3485860.07     10604702.89      3484688.21     10603796.65
      3484255.92     10603468.53      3483880.88     10603202.88
#Sta/Elev= 30
    3352  543.79  3707.6   538.5  4049.9   530.2  4392.2  527.77  4527.1  533.08
  4549.8  530.82  4556.1  527.94  4570.6  528.35  4576.9  525.94  4585.1  527.03
  4591.4  525.08  4599.6   526.4  4605.9   524.8  4620.4   527.4  4626.7  525.33
  4634.9  526.94  4641.2  524.99  4670.2  525.29    4720  528.49  4763.5  524.09
  4969.3  522.63 4972.97  521.54  4991.5  518.08 5046.07  521.57  5048.3  521.93
  5195.8  522.98  5290.1  522.29    5367  523.59  5409.9  523.81  5835.7  534.38
#Mann= 7 ,-1 , 0
    3352     .05       0  4969.3     .04       0  5048.3     .05       0
  5195.8      .1       0  5290.1     .05       0    5367      .1       0
  5409.9     .05       0
#XS Ineff= 2 , 0
       0                 5209.09       0  522.66
Permanent Ineff=
       F       T
Bank Sta=4972.97,5046.07
XS Rating Curve= 0 ,0
Exp/Cntr=0.3,0.1

Type RM Length L Ch R = 1 ,98877   ,753,753,753
BEGIN DESCRIPTION:
PLUMMERS CREEK 105.0
END DESCRIPTION:
XS GIS Cut Line= 4
      3485906.93     10604650.79      3484797.59     10603697.69
      3484464.25     10603567.48      3483887.56     10603136.26
#Sta/Elev= 30
  3298.1   545.6  3584.3  540.74  4123.1  528.75    4336  527.21  4378.8  528.66
  4435.8  532.87  4450.1  531.45    4471  525.26  4485.2  524.02  4620.2  524.49
  4676.2  528.74  4690.4  528.69  4747.5  523.58  4960.5  522.38  4970.5  520.96
  4991.7  516.98  5014.9  520.42  5079.9  521.15  5093.7  522.19    5132  523.16
  5223.7  521.37    5278  521.96  5290.3  522.22  5373.8  523.61  5388.4  525.41
  5395.9  528.01  5410.3  527.57  5438.4  524.58  5473.8  524.98  5838.6  534.81
#Mann= 6 ,-1 , 0
  3298.1     .05       0  4960.5    .035       0  5093.7      .1       0
    5278     .05       0  5290.3      .1       0  5410.3     .05       0
Bank Sta=4970.5,5079.9
XS Rating Curve= 0 ,0
Exp/Cntr=0.3,0.1

Type RM Length L Ch R = 1 ,98124   ,1036,1036,1036
BEGIN DESCRIPTION:
PLUMMERS CREEK 104.0
END DESCRIPTION:
XS GIS Cut Line= 4
      3486255.93     10603473.74      3485271.54     10603338.32
      3484422.59     10602947.69      3483630.93     10602926.86
#Sta/Elev= 30
  3301.1  542.29  3587.6  539.55    3628  539.67  3649.9  540.95  3658.3  538.13
  3678.4  536.72  3860.1  533.09  3880.3   531.1  3961.1  529.68    4010  527.08
  4102.4  524.54  4345.1  522.66  4941.4  520.99  4969.9  520.45  4976.6  519.13
  4998.4  514.95  5009.6  517.58  5044.3  519.11  5061.7     521    5272  523.18
  5359.8   526.9  5479.8  527.89  5709.9  533.31  5809.9  533.07    5880  535.74
    5900  532.45    5930  531.98    5940  532.16    5970  535.78  6021.2  535.99
#Mann= 3 , 0 , 0
  3301.1     .05       0  4976.6    .035       0  5044.3     .05       0
Bank Sta=4976.6,5044.3
XS Rating Curve= 0 ,0
Exp/Cntr=0.3,0.1

Type RM Length L Ch R = 1 ,97088   ,328,328,328
BEGIN DESCRIPTION:
PLUMMERS CREEK 103.0
END DESCRIPTION:
XS GIS Cut Line= 4
       3486563.2     10602025.82      3485396.54     10602187.28
      3484906.96     10602187.28      3484261.11     10602400.82
#Sta/Elev= 30
  3429.1  531.62  3632.1  528.14  3655.6  528.56  3722.4  527.09    3834  526.42
  3924.9  524.24  4019.7  523.25  4086.4  523.16  4106.6  527.43  4116.7  527.52
    4147  523.49  4168.4  522.48  4399.4  519.94  4731.3  517.86  4961.3  518.43
  4971.3  517.63  4991.1  512.01  5021.3  517.19  5031.3   518.3  5091.3  519.77
  5206.9  519.23  5317.5  519.98  5380.9  522.57  5449.6  523.02  5470.2  524.03
  5576.5  524.03  5626.6  524.86  5760.4  526.66  5767.1  526.58  5776.7  526.68
#Mann= 6 ,-1 , 0
  3429.1     .05       0  4961.3     .03       0  5031.3     .05       0
  5626.6     .08       0  5760.4     .05       0  5767.1     .08       0
Bank Sta=4971.3,5021.3
XS Rating Curve= 0 ,0
Exp/Cntr=0.3,0.1

Type RM Length L Ch R = 1 ,96760   ,338,338,338
BEGIN DESCRIPTION:
PLUMMERS CREEK 102.0
END DESCRIPTION:
XS GIS Cut Line= 4
      3486485.05      10601567.5      3485313.21     10602041.44
      3485068.42     10601900.82      3484037.21     10602463.29
#Sta/Elev= 30
  3497.6   530.3  3680.4  528.88  3704.5  530.56  3748.9  527.97  3763.5  530.96
  3787.7  528.11  4201.9  522.95  4353.6  518.78  4813.1  517.11    4931  518.28
  4982.1  516.09  4995.5  512.33  5027.3  516.42  5285.3  519.87  5323.2  518.56
  5426.7   521.9  5448.5  520.46  5519.7  521.65  5535.9  523.87    5645  523.21
  5699.1  525.78  5748.5  524.63  5786.5  526.83  5808.3  525.22  5868.1  528.01
  5895.6   526.8  5949.7  528.68  5977.3  527.42  6037.1  529.59  6218.6  530.43
#Mann= 3 , 0 , 0
  3497.6     .05       0  4982.1    .035       0  5027.3     .08       0
Bank Sta=4982.1,5027.3
XS Rating Curve= 0 ,0
Exp/Cntr=0.3,0.1

Type RM Length L Ch R = 1 ,96422   ,341,341,341
BEGIN DESCRIPTION:
PLUMMERS CREEK 101.0
END DESCRIPTION:
XS GIS Cut Line= 4
      3485974.67     10601223.74        3485308.     10601567.48
      3484938.21     10601754.98       3484184.5     10602077.26
#Sta/Elev= 30
  4099.8  519.95  4151.5  519.14  4195.9  519.91  4234.6   518.2  4456.2  516.41
  4575.2  513.55  4655.6  515.16  4694.3  517.04  4923.8  516.59 4930.07  515.28
  4932.9  514.43  4938.5  515.19  4946.2  513.75  4960.8  513.93  4977.4   510.9
    4991  511.69  5005.1   510.2 5024.82   515.3  5027.6  515.66  5044.3  518.69
  5058.3  519.16  5185.4  518.95  5390.6  520.72  5472.3  520.39  5495.8  521.26
  5572.1     520  5619.1  522.41  5814.9  525.13  5982.2  529.53  6084.2  530.16
#Mann= 4 ,-1 , 0
  4099.8     .08       0  4923.8     .07       0  5027.6     .08       0
  5185.4     .05       0
Bank Sta=4930.07,5024.82
XS Rating Curve= 0 ,0
Exp/Cntr=0.3,0.1

Type RM Length L Ch R = 1 ,96081   ,493,493,493
BEGIN DESCRIPTION:
PLUMMERS CREEK 100.0
END DESCRIPTION:
XS GIS Cut Line= 4
      3485990.31     10601161.23       3485620.5     10601338.32
      3485167.38     10601317.48      3484570.21     10601146.12
#Sta/Elev= 30
  4273.3   519.9  4354.9  518.02  4428.4  517.23  4670.5  516.04  4681.4  515.68
  4711.8  512.74  4731.8  514.27  4771.8  514.48  4791.8  513.33  4811.9  515.18
  4861.9  514.21  4937.3  516.54    4962  516.24    4972  514.43    4982  511.78
  5001.8   510.2  5028.5  514.69  5032.1  515.36  5052.1  516.59    5245  518.29
  5350.5   520.4  5395.5  521.65  5412.9  523.58  5429.3  526.62  5434.5  525.92
    5463   527.2  5496.1  525.54  5527.3  525.63  5574.6  527.93  5758.2  533.43
#Mann= 4 ,-1 , 0
  4273.3     .08       0  4428.4     .05       0    4972    .035       0
  5032.1     .05       0
#XS Ineff= 2 , 0
       0 4917.27  515.88               0
Permanent Ineff=
       T       F
Bank Sta=4972,5028.5
XS Rating Curve= 0 ,0
Exp/Cntr=0.3,0.1

Type RM Length L Ch R = 1 ,95588   ,1061,1061,1061
BEGIN DESCRIPTION:
PLUMMERS CREEK 98.0
END DESCRIPTION:
XS GIS Cut Line= 3
      3486099.64     10601156.01      3485406.96     10600843.53
       3484672.6     10600671.66
#Sta/Elev= 30
  4346.6  521.87  4424.2  519.83  4491.5  518.97  4574.3  515.85  4635.7  515.99
  4710.6   514.2    4780  515.35  4808.6  513.94  4860.4  513.68  4901.1  515.28
  4947.3  515.29  4958.4  513.81  4969.2  512.57    4976  510.57  4990.9  509.28
  5004.6  510.71 5015.75  513.95  5022.3  516.19    5035  519.66    5074  513.65
    5227  514.09  5359.6  517.01  5388.8  519.52  5419.6  519.16  5429.9  520.87
  5439.4  521.13  5444.6  520.11  5450.4  521.15  5577.2  524.12  5860.7  534.34
#Mann= 4 ,-1 , 0
  4346.6     .08       0  4424.2     .05       0  4947.3    .035       0
  5022.3     .05       0
#XS Ineff= 2 , 0
       0 4934.32  515.78               0
Permanent Ineff=
       T       F
Bank Sta=4958.4,5015.75
XS Rating Curve= 0 ,0
Exp/Cntr=0.3,0.1

Type RM Length L Ch R = 1 ,94527   ,1365,1365,1365
BEGIN DESCRIPTION:
PLUMMERS CREEK 96.0
END DESCRIPTION:
XS GIS Cut Line= 3
      3486917.36      10600390.4      3485604.88     10600171.65
      3484651.76     10600020.61
#Sta/Elev= 30
    4107  527.25  4676.1  516.85  4710.5  518.06    4742  512.96  4791.6  513.65
  4811.8  517.73  4863.7  513.06  4974.1  512.93  4977.3  511.46  4994.1  507.76
 5021.88  511.51  5024.7  511.92  5085.6  515.25  5278.2  513.51  5659.7   518.6
    5722   516.1  5754.3   517.9  5794.8  531.43  5804.9   531.6  5851.7  523.68
  5895.1   523.3  5958.2  524.07  6098.5  532.21  6118.8  539.95  6128.9  540.38
  6159.3  536.38  6199.8  535.21  6260.5   537.3  6311.1  542.83  6402.6  542.47
#Mann= 5 ,-1 , 0
    4107     .05       0  4974.1    .035       0  5024.7     .05       0
  5895.1     .08       0  5958.2     .05       0
Bank Sta=4977.3,5021.88
XS Rating Curve= 0 ,0
Exp/Cntr=0.3,0.1

Type RM Length L Ch R = 1 ,93162   ,1220,1220,1220
BEGIN DESCRIPTION:
PLUMMERS CREEK 93.0
END DESCRIPTION:
XS GIS Cut Line= 4
      3487698.65     10598645.61      3486537.17     10598879.98
      3485688.21     10599171.65      3484828.87     10599213.32
#Sta/Elev= 30
    3119  531.54  3258.3  529.61  3376.6  525.54  3579.4  521.18    3646  518.45
  3941.8  514.85  3972.4  513.81  3992.8  510.58  4013.2  513.92  4036.5  514.79
  4436.1  510.77  4827.4  509.54  4881.9  511.16  4907.9  508.17  4954.2   510.1
  4970.4  509.19  5001.4  504.34  5049.4  509.27  5070.6  510.01  5237.7  515.59
  5277.7  513.04  5287.8  517.76  5308.7  520.38  5327.8  515.04  5337.8  514.35
  5417.9  515.04    5518  524.36  5668.2  525.81  5888.5  533.94  6061.9  537.45
#Mann= 4 ,-1 , 0
    3119     .08       0  3376.6     .05       0  4954.2    .035       0
  5070.6     .05       0
Bank Sta=4970.4,5049.4
XS Rating Curve= 0 ,0
Exp/Cntr=0.3,0.1

Type RM Length L Ch R = 1 ,91942   ,1658,1658,1658
BEGIN DESCRIPTION:
PLUMMERS CREEK 90.0
END DESCRIPTION:
XS GIS Cut Line= 4
      3488136.11     10597984.15      3486834.04     10597968.53
      3485828.84     10598239.36      3485172.59     10598406.03
#Sta/Elev= 30
  2927.3  537.96  3041.3  538.75  3194.1  535.52  3271.3  534.61  3331.3  538.07
  3401.3  537.62  3481.3  531.66  3741.4  528.75  3931.4  523.85  3981.4  521.04
  4051.4  521.44  4448.3  510.36  4542.2  510.26  4568.1  508.74  4738.9  507.63
  4925.4  508.09  4935.7  506.77  4977.1  508.13 4987.46  506.84  4997.9  501.75
    5008  501.12  5011.2  501.62 5020.12  506.83  5026.6  508.26  5173.9  509.21
  5383.6  513.32  5638.6  521.09  5772.7  527.62  5910.7  532.55  5947.6  532.83
#Mann= 4 ,-1 , 0
  2927.3     .08       0  3194.1     .05       0  4977.1     .03       0
  5026.6     .05       0
Bank Sta=4987.46,5020.12
XS Rating Curve= 0 ,0
Exp/Cntr=0.3,0.1

Type RM Length L Ch R = 1 ,90284   ,996,996,996
BEGIN DESCRIPTION:
PLUMMERS CREEK 88.0
END DESCRIPTION:
XS GIS Cut Line= 4
      3488209.02     10596593.53      3487172.59     10596567.48
      3485797.59     10596895.61      3484120.55       10596255.
#Sta/Elev= 30
  2973.8  541.23  3030.7     539  3590.9  530.99  4222.1  518.92  4617.6  513.11
  4695.5  510.22    4869   507.2 4909.33  503.57    4926     502  4946.6  502.92
  4966.9  500.09  4987.7  502.38  5008.3  501.36 5025.28  503.69  5037.4  504.89
  5042.6  503.95  5141.9  504.08  5384.5  506.22  5672.2  506.74  5708.4  506.53
  5740.5  502.97  5762.4  502.87    5794  504.79  5911.8  506.92  5951.5  509.04
  6104.4  508.97    6158  511.12  6345.7  513.14  6909.6  527.35  7219.4  531.86
#Mann= 3 , 0 , 0
  2973.8     .05       0 4909.33     .03       0 5025.28     .05       0
#XS Ineff= 2 , 0
       0                 5702.27       0  504.94
Permanent Ineff=
       F       T
Bank Sta=4909.33,5025.28
XS Rating Curve= 0 ,0
Exp/Cntr=0.3,0.1

Type RM Length L Ch R = 1 ,89288   ,213,213,213
BEGIN DESCRIPTION:
PLUMMERS CREEK 87.0
END DESCRIPTION:
XS GIS Cut Line= 4
      3488167.39     10596249.78      3487136.13     10596135.19
        3485933.     10595775.82      3484880.96     10595489.37
#Sta/Elev= 30
  3028.9   541.7  3111.7   539.9  3798.9  526.02  4201.2  520.34  4415.6  515.64
  4456.9  513.56    4691  510.65  4853.4   507.1  4938.5  503.18  4947.4   502.4
  4988.9  498.93  5020.4  501.16  5037.9  500.75  5043.1  501.69  5083.1  500.43
  5109.4  502.39  5135.2  503.05  5175.6  501.78  5208.3  502.19  5530.4  508.74
  5571.8  510.03  5592.6  511.98  5626.2  511.38  5675.5  515.09    5862  524.76
    5976  528.62  6069.3  528.82  6117.2  526.81  6172.9  526.62  6412.5  531.81
#Mann= 4 ,-1 , 0
  3028.9      .1       0  3111.7     .05       0  4938.5     .03       0
  5135.2     .05       0
Bank Sta=4947.4,5109.4
XS Rating Curve= 0 ,0
Exp/Cntr=0.3,0.1

Type RM Length L Ch R = 1 ,89075   ,257,257,257
BEGIN DESCRIPTION:
PLUMMERS CREEK 86.0
END DESCRIPTION:
XS GIS Cut Line= 4
      3488183.05     10596124.79      3486604.88     10595713.32
      3485537.17     10595572.69      3484725.94     10595380.28
#Sta/Elev= 30
  3082.8  541.46  3187.2  539.94  3314.8  537.98  3838.2  525.35  3982.4  524.57
  4168.9  518.63  4478.9  513.74  4571.9  509.85  4619.9  510.75  4827.5  507.06
  4968.7  502.74 4971.34  501.98  4988.6  498.88  5019.1  502.04  5029.2  502.42
  5099.8  502.39  5140.2  500.87  5160.3     503  5200.7  501.01  5261.2  503.23
  5382.4  503.93  5608.2  509.29  5681.8  512.09  5945.9  526.79    6022  529.11
  6209.5  526.61  6293.9  527.65  6378.4  530.63  6525.6  529.88  6624.4  531.71
#Mann= 4 ,-1 , 0
  3082.8      .1       0  3187.2     .05       0  4968.7     .04       0
  5029.2     .05       0
Bank Sta=4971.34,5019.1
XS Rating Curve= 0 ,0
Exp/Cntr=0.3,0.1

Type RM Length L Ch R = 1 ,88818   ,299,299,299
BEGIN DESCRIPTION:
PLUMMERS CREEK 85.0
END DESCRIPTION:
XS GIS Cut Line= 4
      3488172.58     10595843.53      3486906.96     10595484.15
      3485781.96     10595379.98      3484532.71     10595036.44
#Sta/Elev= 30
  3071.1   543.7  3123.6  542.83  3242.5  538.36  3328.6  535.73  3388.9  533.43
  3705.7   527.9  3736.9  525.62  3809.7  525.45  4191.8  513.98  4601.6  508.53
  4733.1  506.61  4773.3  503.93  4853.6  503.99  4974.1   501.6  4984.2   500.2
  5014.7  493.02  5034.4  497.95  5064.5  500.25  5119.4   501.7    5185  501.28
  5447.8  506.77    5639   511.6  5837.9  518.49  6014.2  521.22  6127.9  522.06
    6133  521.27  6449.8  524.89  6480.9  523.36  6582.3  527.61  6812.2  529.61
#Mann= 6 ,-1 , 0
  3071.1      .1       0  3242.5     .08       0  3328.6     .05       0
  4601.6     .08       0  4974.1     .07       0  5119.4     .08       0
Bank Sta=4984.2,5064.5
XS Rating Curve= 0 ,0
Exp/Cntr=0.3,0.1

Type RM Length L Ch R = 1 ,88519   ,1235,1235,1235
BEGIN DESCRIPTION:
PLUMMERS CREEK 84.0
END DESCRIPTION:
XS GIS Cut Line= 4
      3488125.71     10595546.65      3487198.63     10595301.86
      3485823.63     10595083.11      3484407.04     10594723.76
#Sta/Elev= 30
  3091.9  543.64  3416.3  532.08  4031.8  514.69  4563.6  504.96    4756  503.08
  4787.8  504.67  4826.9  501.99  4948.4  501.94  4958.6  499.89  4979.2  493.09
  5009.2  499.97  5201.6  502.82  5233.3  500.77  5357.7  501.62  5383.8  503.85
  5404.1  501.85  5419.9  504.32    5425  502.09  5454.9  506.36  5537.5  507.93
  5587.6  504.06  5609.7   507.4  5633.8  505.74  5702.5   509.8  5915.4  515.46
  6218.4   519.3  6249.3  516.57  6311.2  516.54  6507.2  525.76  6904.5  530.86
#Mann= 3 , 0 , 0
  3091.9     .05       0  4958.6    .035       0  5009.2     .05       0
Bank Sta=4958.6,5009.2
XS Rating Curve= 0 ,0
Exp/Cntr=0.3,0.1

Type RM Length L Ch R = 1 ,87284   ,1245,1245,1245
BEGIN DESCRIPTION:
PLUMMERS CREEK 82.0
END DESCRIPTION:
XS GIS Cut Line= 4
      3487943.38     10594442.47      3487505.92     10594249.78
      3486255.92     10593989.36      3485287.14     10593921.65
#Sta/Elev= 30
  3812.1  541.84  3868.1  536.36  3933.7  537.58    4200  525.45  4228.8  521.91
  4334.9   516.4  4453.9  513.81  4477.9  511.06  4597.5  507.09    4672  507.05
  4712.8  502.75  4867.5   499.9  4968.2  500.37 4974.33  497.75  4998.6  491.26
  5029.5  497.54  5060.1  499.16  5092.9  500.97  5182.7   499.4  5274.6  505.43
  5366.6  502.83  5433.1  508.64  5533.2  508.68  5566.3  513.23    5641  512.28
  5691.1  516.21  5761.2  512.96  5894.7  521.73  5941.7  520.82  6538.1  538.24
#Mann= 6 ,-1 , 0
  3812.1     .05       0  4453.9     .16       0  4867.5     .05       0
  4968.2     .05       0  4968.2     .03       0  5060.1     .05       0
Bank Sta=4974.33,5029.5
XS Rating Curve= 0 ,0
Exp/Cntr=0.3,0.1

Type RM Length L Ch R = 1 ,86039   ,795,795,795
BEGIN DESCRIPTION:
PLUMMERS CREEK 79.0
END DESCRIPTION:
XS GIS Cut Line= 2
      3488146.57     10593864.39      3486531.97     10592109.16
#Sta/Elev= 30
  3956.6  534.21  4060.7  535.21  4082.3  533.22  4110.1  534.13  4195.1  531.16
  4351.1  523.32  4634.1  505.42  4761.7  501.27  4938.6  497.86  4959.6     497
 4963.37  495.95  4973.8  494.51  4980.6  494.71  4994.8  490.22  5001.9  489.45
  5005.2  489.95  5016.3  494.69  5023.1  495.64  5030.5  497.92  5037.3  498.54
  5136.6  497.11  5426.9  503.82  5447.9  506.08    5533  508.54    5837  521.83
  5992.9  527.47    6099  533.97  6176.7  537.49  6240.8  539.98  6341.5  541.35
#Mann= 3 , 0 , 0
  3956.6     .05       0 4963.37     .03       0  5023.1     .05       0
Bank Sta=4963.37,5023.1
XS Rating Curve= 0 ,0
Exp/Cntr=0.3,0.1

Type RM Length L Ch R = 1 ,85244   ,1362,1362,1362
BEGIN DESCRIPTION:
PLUMMERS CREEK 77.0
END DESCRIPTION:
XS GIS Cut Line= 4
      3489084.04     10592416.44      3488417.38     10592416.44
       3487495.5     10592406.03      3486990.33     10591911.27
#Sta/Elev= 30
  3648.1  526.37    3720   525.5    3910  520.72    4000  519.47    4050  517.08
    4120  515.23    4160  512.98    4220  511.35    4290  507.51    4360  504.74
  4870.1  496.39  4930.1  495.54  4960.1  496.02  4980.1  494.18  4990.1  491.21
  4997.1  487.79  4999.8  487.29  5010.1  488.98  5025.5   494.3  5030.1  495.34
  5040.1  495.75  5130.1  495.28  5210.1  498.04  5298.7  503.24  5390.7  511.38
  5433.2  513.53  5553.3  523.66  5638.2  529.11  5822.1  537.19  5943.8  541.63
#Mann= 3 , 0 , 0
  3648.1     .05       0  4980.1    .035       0  5025.5     .05       0
Bank Sta=4980.1,5025.5
XS Rating Curve= 0 ,0
Exp/Cntr=0.3,0.1

Type RM Length L Ch R = 1 ,83882   ,723,723,723
BEGIN DESCRIPTION:
PLUMMERS CREEK 74.0
END DESCRIPTION:
XS GIS Cut Line= 2
        3489125.     10591399.77      3486911.46     10591004.81
#Sta/Elev= 30
  3946.2  521.57  4335.1  517.37  4446.9   517.2  4639.9  513.66  4822.9   503.3
  4876.7  499.02  4930.6  493.21  4975.1  492.18 4978.18  491.19  4984.5  489.22
  4989.5  489.96  4992.4  484.72  4995.2  484.22  5005.6  485.24  5015.7  489.63
 5024.21  491.15    5036   492.7  5102.3  491.56  5161.3  492.99  5215.1  495.93
  5391.9  499.46  5558.6  505.83  5706.5  513.67  5730.3  513.82  5777.6  517.65
  5789.3  517.25  5843.1  522.44  5980.7  530.54  6068.7  537.39  6194.7  543.44
#Mann= 3 , 0 , 0
  3946.2     .05       0 4978.18     .03       0 5024.21     .05       0
Bank Sta=4978.18,5024.21
XS Rating Curve= 0 ,0
Exp/Cntr=0.3,0.1

Type RM Length L Ch R = 1 ,83159   ,1022,1022,1022
BEGIN DESCRIPTION:
PLUMMERS CREEK 72.0
END DESCRIPTION:
XS GIS Cut Line= 4
      3489116.38      10590635.9       3488617.2     10590470.96
      3487419.29      10590583.8      3486812.99     10590757.03
#Sta/Elev= 30
  3766.5  514.56  4202.8   509.2  4317.4  506.18  4352.7  503.37  4648.9  497.83
  4776.9  494.83  4885.4   490.9  4970.3     491  4980.3  489.45    4989  483.67
    4994  483.39  5000.2  481.39  5003.4  481.89  5010.5   486.3  5020.5  488.22
  5040.6  490.02  5110.9  491.13  5206.1  495.47  5251.5  498.91  5309.6  505.17
  5314.6     505    5352  508.98  5418.2  514.31  5613.5  525.56  5764.3  530.81
  5909.9  533.57  5977.5   533.4  6016.5  534.36  6123.1  533.71    6126  534.45
#Mann= 3 , 0 , 0
  3766.5     .05       0  4980.3    .035       0  5040.6     .05       0
Bank Sta=4980.3,5040.6
XS Rating Curve= 0 ,0
Exp/Cntr=0.3,0.1

Type RM Length L Ch R = 1 ,82137   ,175,175,175
BEGIN DESCRIPTION:
PLUMMERS CREEK 71.0
END DESCRIPTION:
XS GIS Cut Line= 3
      3489051.24     10590392.84      3488725.71     10589906.72
      3487657.96     10589377.19
#Sta/Elev= 30
  3963.9  511.41  4085.7  508.87  4166.5     508  4181.5  507.18  4295.6  506.57
  4367.6  503.98  4505.7  502.54  4541.7  501.41  4637.9  495.88  4854.4  489.81
  4890.1   487.3  4929.3  487.45  4951.7  488.97  4974.2  488.69  4979.7  487.74
  4993.6  481.05  4996.3  480.55    5019  486.33    5033  487.61  5069.4  489.92
  5108.7  489.89  5220.7  493.62  5265.6  496.08  5310.4  498.87  5390.1  505.17
  5467.3  509.69  5489.7  511.75  5501.8  513.71  5534.6  514.16  5740.8  521.51
#Mann= 3 , 0 , 0
  3963.9     .05       0  4979.7    .035       0    5033     .05       0
Bank Sta=4979.7,5033
XS Rating Curve= 0 ,0
Exp/Cntr=0.3,0.1

Type RM Length L Ch R = 1 ,81962   ,253,253,253
BEGIN DESCRIPTION:
PLUMMERS CREEK 70.0
END DESCRIPTION:
XS GIS Cut Line= 4
      3489198.79     10590340.73      3488717.03     10589720.09
      3488152.79     10589424.95      3487397.56     10589073.37
#Sta/Elev= 30
  3896.1  512.46  4078.4  508.14  4256.7   505.6    4292  505.84    4435  502.92
  4598.8  501.63  4663.1  499.68  4707.5  496.45  4823.5  492.69  4867.9  490.15
  4972.4   487.5  4980.8  486.29  4994.5  480.97  5003.1  480.02  5006.3  480.52
  5016.5  485.23  5055.1  487.35  5082.8  488.81  5231.6  492.59    5308  497.17
  5396.5  504.34  5456.9  508.25  5485.3  511.33  5576.8  513.43  5668.4  518.06
  5771.6  521.03  5788.3   522.3  5925.5  524.84  5959.4  524.56  6151.6  528.54
#Mann= 3 , 0 , 0
  3896.1     .05       0  4972.4    .035       0  5055.1     .05       0
Bank Sta=4972.4,5055.1
XS Rating Curve= 0 ,0
Exp/Cntr=0.3,0.1

Type RM Length L Ch R = 1 ,81709   ,305,305,305
BEGIN DESCRIPTION:
PLUMMERS CREEK 69.1
END DESCRIPTION:
XS GIS Cut Line= 4
      3488990.47      10589763.5      3488773.45     10589403.25
      3488404.53     10589307.76      3487945.79      10588970.2
#Sta/Elev= 30
  4302.8  501.88  4362.5  500.41  4383.8   501.2  4417.1  500.72  4572.1  498.53
  4596.9  498.44  4776.4  494.91  4831.4  492.11  4953.2  491.66  4972.7  489.84
 4977.22  487.17  4988.7  480.39  4993.6  479.53  5003.7  480.23    5014   482.7
  5024.1  486.38  5034.6  487.13    5045  486.15    5076  487.95  5189.4  491.69
  5195.6  492.62  5204.1  492.28  5211.2  493.41  5239.6  494.02  5260.4  496.13
  5396.2  503.52  5525.5  511.85  5609.4  515.05  5644.8  515.45    5674  516.11
#Mann= 11 ,-1 , 0
  4302.8     .15       0  4417.1     .08       0  4572.1     .15       0
  4596.9     .05       0  4972.7     .03       0  5034.6     .05       0
  5211.2     .08       0  5396.2     .05       0  5525.5     .08       0
  5609.4     .05       0  5644.8     .08       0
Bank Sta=4977.22,5034.6
XS Rating Curve= 0 ,0
Exp/Cntr=0.3,0.1

Type RM Length L Ch R = 1 ,81404   ,446,446,446
BEGIN DESCRIPTION:
PLUMMERS CREEK 69.0
END DESCRIPTION:
XS GIS Cut Line= 4
      3489046.89     10589720.08      3488847.24     10589294.74
      3488539.08     10588921.48      3488036.37     10588687.46
#Sta/Elev= 30
  4317.5  501.08  4415.9  499.62  4478.8  499.45  4514.6  498.25    4630  496.35
  4821.4  493.91  4850.1  491.32  4913.9  491.89  4963.4  488.91  4971.3  486.37
  4985.6  481.08  4991.8  480.18  5006.4  481.97  5020.7   485.9  5027.2  486.37
  5076.7  486.77  5119.7  488.79  5247.4  495.01  5278.2  497.12  5283.7  498.24
  5301.1  498.27  5306.6  499.61  5329.5  497.99    5335  499.09  5375.2  499.59
    5615  508.86  5698.2  510.25  5729.4  512.39  5757.8  512.07  5825.9   513.1
#Mann= 4 ,-1 , 0
  4317.5     .15       0    4630     .05       0  4963.4     .03       0
  5119.7     .05       0
Bank Sta=4971.3,5027.2
XS Rating Curve= 0 ,0
Exp/Cntr=0.3,0.1

Type RM Length L Ch R = 1 ,80958   ,80,80,80
BEGIN DESCRIPTION:
PLUMMERS CREEK 68.1
END DESCRIPTION:
XS GIS Cut Line= 3
      3489220.51     10589806.93      3489090.29     10588778.25
      3488352.48     10588374.62
#Sta/Elev= 30
  4146.2  504.01  4282.6  499.13  4335.3  499.47  4434.5  497.92    4595  494.83
  4725.9  490.82  4867.6   489.6  4971.3  490.38  4978.1  489.84  4988.2  487.48
 4993.61  484.62  4998.2  482.04  5008.1  479.33  5018.4  479.96  5028.5  484.37
    5089  488.03  5169.6  491.31    5252  491.98    5290  489.66  5340.6  490.24
  5349.7  491.52  5355.4   493.6  5386.2  495.92  5687.4  501.12  5774.7  503.52
  5834.4  503.41  5856.2  504.52  5864.9  503.52    5878  503.71  6024.1  507.55
#Mann= 5 ,-1 , 0
  4146.2     .15       0  4434.5      .1       0  4867.6     .05       0
  4988.2     .03       0  5028.5     .05       0
Bank Sta=4993.61,5028.5
XS Rating Curve= 0 ,0
Exp/Cntr=0.3,0.1

Type RM Length L Ch R = 1 ,80878   ,293,293,293
BEGIN DESCRIPTION:
PLUMMERS CREEK 68.0
END DESCRIPTION:
XS GIS Cut Line= 4
      3489346.38     10589841.66      3489211.82       10589247.
       3489177.1     10588721.82      3488669.26     10588079.43
#Sta/Elev= 30
  4106.1   503.2  4137.8  502.66  4371.1  497.71  4413.7  497.66  4434.2  496.71
  4471.3  496.19  4645.5  492.46  4751.2  490.79  4771.3  489.52  4831.5  488.78
  4871.5  488.08  4937.8  484.91  4942.8  485.72  4971.7  484.63  4981.7  484.75
  4991.8  482.99  4998.8  478.77  5001.5  478.27  5011.8  478.92  5021.8   483.3
  5031.8  484.42  5142.1  489.61  5202.7  490.74  5239.7   490.5  5257.8  491.03
  5439.9  493.23  5609.3  494.25  5673.4  495.33  5965.2  496.92    6061  498.41
#Mann= 8 ,-1 , 0
  4106.1      .1       0  4137.8     .15       0  4471.3      .1       0
  4831.5     .05       0  4981.7     .03       0  5031.8     .05       0
  5202.7     .08       0  5257.8     .05       0
Bank Sta=4981.7,5031.8
XS Rating Curve= 0 ,0
Exp/Cntr=0.3,0.1

Type RM Length L Ch R = 1 ,80585   ,245,245,245
BEGIN DESCRIPTION:
PLUMMERS CREEK 67.0
END DESCRIPTION:
XS GIS Cut Line= 4
      3489546.02     10589520.41       3489489.6     10589151.51
      3489476.58     10588786.93      3489221.23     10588345.47
#Sta/Elev= 30
  4416.5  498.18  4478.2  496.73  4546.8  494.51  4628.9   492.7  4786.1   489.9
  4839.6  488.52  4919.6  482.98  4929.7  482.68  4959.7  484.06  4969.7  483.74
  4979.7  483.28  4989.7  481.07  4996.7  478.45  4999.4  477.95  5002.7  478.45
  5009.7  478.47  5019.7  480.54  5029.7  483.65  5039.7  484.26  5059.7  483.95
  5079.7  484.18  5089.8  484.75  5119.8  487.73  5137.3   488.4  5206.8  488.97
  5234.5  488.44  5299.2  489.18  5553.3  490.04  5634.9  490.97  5664.5  491.18
#Mann= 7 ,-1 , 0
  4416.5     .05       0  4628.9     .08       0  4786.1     .05       0
  4959.7     .03       0  5039.7     .05       0  5553.3     .08       0
  5634.9     .05       0
Bank Sta=4969.7,5029.7
XS Rating Curve= 0 ,0
Exp/Cntr=0.3,0.1

Type RM Length L Ch R = 1 ,80340   ,917,917,917
BEGIN DESCRIPTION:
PLUMMERS CREEK 66.3
END DESCRIPTION:
XS GIS Cut Line= 4
      3489650.18     10589494.42      3489819.46     10589086.41
      3489567.73     10588565.57      3489156.31     10588067.54
#Sta/Elev= 30
    4308   497.4  4326.7  497.21  4350.5  495.88  4440.9  494.38    4510   492.4
  4527.5  492.42  4581.6  490.53  4646.6  489.11  4887.9  486.61    4916  485.61
  4938.6  483.75  4977.2  481.77  4989.4  478.59  4999.1  477.11    5012  480.27
  5021.6  481.71  5043.8  483.06  5096.8  482.62  5154.9  485.67  5199.3  487.12
  5232.4  487.09  5237.9  487.54  5260.5  487.03  5266.1  487.72  5305.7  487.47
  5348.8  488.32  5505.2   489.3  5718.8  489.94    5939  491.49  5974.2  492.21
#Mann= 3 , 0 , 0
    4308     .05       0  4977.2     .03       0  5021.6     .05       0
Bank Sta=4977.2,5021.6
XS Rating Curve= 0 ,0
Exp/Cntr=0.3,0.1

Type RM Length L Ch R = 1 ,79423   ,457,457,457
BEGIN DESCRIPTION:
PLUMMERS CREEK 66.2
END DESCRIPTION:
XS GIS Cut Line= 4
       3491096.9     10589320.59      3490473.86     10588532.64
      3490171.52     10588042.47      3489154.56       10587676.
#Sta/Elev= 30
  3579.2  500.95  3773.9  497.23  4030.4  488.08  4222.7  483.35  4400.6  481.66
  4514.4   482.7  4564.1  481.52  4678.9  476.65  4730.8  476.21  4752.1  475.05
  4767.5  477.87  4819.6  479.33  4941.3  479.38  4956.7  478.44  4962.6  476.65
  4972.1  475.72  4993.4  470.41  5007.6  468.51  5014.7  470.54 5026.68  476.48
    5036  479.25  5181.2  485.25  5307.8  485.05  5466.9  486.26  5502.9  484.61
  5620.3  484.56  6041.2  489.67  6120.8  490.95  6158.2   492.7  6240.6  492.43
#Mann= 3 ,-1 , 0
  3579.2     .05       0  4956.7     .03       0    5036     .05       0
#XS Ineff= 1 ,-1
  4528.4 4813.74  480.23
Permanent Ineff=
       F
Bank Sta=4962.6,5026.68
XS Rating Curve= 0 ,0
Exp/Cntr=0.3,0.1

Type RM Length L Ch R = 1 ,78966   ,229,229,229
BEGIN DESCRIPTION:
PLUMMERS CREEK 66.1
END DESCRIPTION:
XS GIS Cut Line= 4
      3491303.81      10589012.6      3490769.98     10588444.05
      3490618.07     10587966.62      3488835.69     10587151.32
#Sta/Elev= 30
  3946.7  497.78  4309.3  486.99  4401.2  483.32  4599.4  482.27  4767.4  478.22
    4876     479  4971.3  476.39    4981  474.93  4998.3  469.26  5012.2  468.76
  5035.8  476.36  5043.9  477.94  5054.4  478.21  5117.4  477.06  5234.2  478.37
  5325.7  476.83  5509.1  479.53  5566.8  478.79  5779.5  483.37  6026.1  480.58
  6256.3  485.18  6284.8  484.64  6313.3  480.56  6376.9  483.85  6410.9  483.16
  6451.4  484.13    6526  488.71  6554.5  489.34  6751.7  492.28  7187.6  495.68
#Mann= 3 , 0 , 0
  3946.7     .05       0  4971.3     .03       0  5035.8     .05       0
Bank Sta=4971.3,5035.8
XS Rating Curve= 0 ,0
Exp/Cntr=0.3,0.1

Type RM Length L Ch R = 1 ,78737   ,1202,1202,1202
BEGIN DESCRIPTION:
PLUMMERS CREEK 66.0
END DESCRIPTION:
XS GIS Cut Line= 4
      3491651.05     10588778.24      3490978.32     10588140.23
      3490466.16     10587710.54      3488782.13     10586829.46
#Sta/Elev= 30
  3929.2  496.29  4074.7   494.9  4463.8  484.65  4923.7  479.98  4966.6     477
  4973.1   475.6  4980.9  474.45  4987.4  471.22  5001.5  469.35  5016.1  470.66
  5030.4  474.77  5036.9  477.03  5215.1  476.71  5371.2  478.06  5420.6  476.35
    5491  477.54  5631.1  475.73  5876.1  482.07  6008.5  479.42  6201.5  481.49
  6207.1  480.27  6223.6  479.69  6229.2   477.1    6240  476.83  6251.8  478.95
  6267.7  480.01  6350.4   483.9  6587.5  488.64  7133.7  493.78  7425.5  499.26
#Mann= 3 ,-1 , 0
  3929.2     .05       0  4966.6    .035       0  5036.9     .05       0
#XS Ineff= 2 , 0
       0                 5045.45       0  477.57
Permanent Ineff=
       F       T
Bank Sta=4973.1,5030.4
XS Rating Curve= 0 ,0
Exp/Cntr=0.3,0.1

Type RM Length L Ch R = 1 ,77535   ,2224,2224,2224
BEGIN DESCRIPTION:
PLUMMERS CREEK 63.2
END DESCRIPTION:
XS GIS Cut Line= 4
      3492453.97     10587319.91      3491494.81      10587146.3
      3490939.25     10586868.53      3489286.38     10586881.54
#Sta/Elev= 30
  3688.1  487.17  4015.2   482.9  4100.5  483.14  4167.6  485.16    4266  482.93
  4756.2   480.5    4773  481.14  4884.8  478.12  4912.7  476.72  4951.9  472.68
  4957.5  472.12  4967.7  469.56  4979.8   469.3  4990.1  467.74  5001.9  464.85
  5005.2  465.35 5018.82  472.28    5019  473.09  5034.8  473.96  5091.6   472.4
  5213.7  473.85  5401.1   473.2  5491.1  474.53  5581.1  474.43  5641.1  475.84
  5761.1   474.1  5801.1  470.38  5851.1  473.88  5921.1   476.3  6936.9  490.66
#Mann= 3 ,-1 , 0
  3688.1     .05       0  4951.9     .03       0    5019     .05       0
#XS Ineff= 1 ,-1
 5654.56 6019.81  475.25
Permanent Ineff=
       F
Bank Sta=4957.5,5018.82
XS Rating Curve= 0 ,0
Exp/Cntr=0.3,0.1

Type RM Length L Ch R = 1 ,75311   ,777,777,777
BEGIN DESCRIPTION:
PLUMMERS CREEK 63.1
END DESCRIPTION:
XS GIS Cut Line= 4
      3491434.07      10586304.3      3490817.73      10586143.7
      3490266.51     10585753.07      3489220.54     10585466.63
#Sta/Elev= 30
  3881.4  479.86  4386.1  472.35  4682.3  471.42  4732.8  469.74  4789.3  470.84
  4860.7   468.9  4946.8  469.68 4956.18  468.29  4967.7  465.01    4991  463.34
  5003.2  460.61  5029.5  468.31    5040  469.63    5140  469.75    5330  477.93
  5404.1  479.27  5631.7  478.37  5711.1  474.57  5727.3  475.11  5750.7  471.59
  5779.1   474.3  5785.2  475.81  5819.7  475.64  5865.6  477.84  5978.4  480.56
  6027.9  479.95  6052.5  481.17    6087  485.18  6126.7  488.15  6278.4  495.01
#Mann= 5 ,-1 , 0
  3881.4     .05       0  4946.8    .035       0    5040     .05       0
  5819.7     .16       0  5865.6     .05       0
Bank Sta=4956.18,5029.5
XS Rating Curve= 0 ,0
Exp/Cntr=0.3,0.1

Type RM Length L Ch R = 1 ,74534   ,1615,1615,1615
BEGIN DESCRIPTION:
PLUMMERS CREEK 63.0
END DESCRIPTION:
XS GIS Cut Line= 3
      3491447.07     10585687.97      3490314.25     10585210.54
      3489758.69     10584928.42
#Sta/Elev= 30
  4317.3  481.74  4355.2  479.19  4448.5  475.62  4572.3   475.9  4843.6  473.44
  4854.4  472.48 4864.22  467.64  4876.1  463.81  4884.4  462.67  4908.1  464.41
  4973.8  464.53  4984.6  462.56  4995.3  459.03  5006.4  460.77 5017.16   467.6
  5019.3  468.86  5028.1  468.87  5212.5  467.06  5219.9  465.45  5225.4  462.52
  5234.2  461.05  5255.9  465.88  5272.8  467.25  5455.2  468.21  5571.5  471.24
  5666.2  474.93    5733  478.82  5860.9  490.94  6000.1  501.14  6169.7  505.95
#Mann= 3 , 0 , 0
  4317.3     .05       0 4864.22     .07       0 5017.16     .05       0
Bank Sta=4864.22,5017.16
XS Rating Curve= 0 ,0
Exp/Cntr=0.3,0.1

Type RM Length L Ch R = 1 ,72919   ,1387,1387,1387
BEGIN DESCRIPTION:
PLUMMERS CREEK 62.0
END DESCRIPTION:
XS GIS Cut Line= 6
      3491481.79     10585627.22      3491164.95     10584945.78
      3490431.44     10584507.42      3489541.68      10584225.3
      3489559.04       10584247.      3489368.06     10584194.91
#Sta/Elev= 30
  3649.1  480.48  3688.9  477.53    3872  478.13  4074.3   474.9  4203.4  473.77
  4239.7  474.55  4261.8  473.03    4361  470.74  4472.4  469.84  4515.2  467.62
  4683.5  467.15  4733.1  465.05  4785.6  466.64  4858.2  465.85    4881  458.81
  4902.4  461.01  4945.2  461.66  4966.6  464.63  4974.7  463.57  4982.1  460.67
  4997.5  457.65  5040.5  466.06  5091.2  467.82  5258.7  471.54  5323.2  476.56
  5489.9  484.29  5651.3  495.32  5925.8  508.79  6081.4  512.79  6415.6  515.29
#Mann= 3 ,-1 , 0
  3649.1     .05       0  4515.2     .07       0  5091.2     .05       0
Bank Sta=4858.2,5040.5
XS Rating Curve= 0 ,0
Exp/Cntr=0.3,0.1

Type RM Length L Ch R = 1 ,71532   ,1463,1463,1463
BEGIN DESCRIPTION:
PLUMMERS CREEK 60.0
END DESCRIPTION:
XS GIS Cut Line= 4
       3491894.1     10584793.86      3491581.61     10584481.37
      3491403.66     10583795.61        3490770.     10583240.07
#Sta/Elev= 30
    4208  475.89  4225.1  475.32  4295.8  476.44    4416  476.09  4486.7  474.56
  4500.9  475.23  4610.6  469.41  4671.7  466.61  4747.6  465.64  4773.6  463.22
  4828.8  464.12  4904.8  463.11  4945.3  465.11  4959.6  463.48  4980.2  462.77
  4985.9  458.04  5000.7   453.7  5011.2  456.63  5052.6  459.76  5073.2  463.74
  5124.9  462.94  5217.9  465.44  5369.6   467.4  5525.2  469.29  5780.5  479.34
  5844.1  483.89    5901  486.04  6035.8  496.11    6106  503.43  6201.1  508.55
#Mann= 5 ,-1 , 0
    4208     .05       0  4610.6      .1       0  4747.6     .07       0
  5217.9     .16       0  5369.6     .05       0
Bank Sta=4959.6,5073.2
XS Rating Curve= 0 ,0
Exp/Cntr=0.3,0.1

Type RM Length L Ch R = 1 ,70069   ,1779,1779,1779
BEGIN DESCRIPTION:
PLUMMERS CREEK 58.0
END DESCRIPTION:
XS GIS Cut Line= 3
      3492263.04     10584429.28      3492141.51       10583622.
      3491273.42     10582979.61
#Sta/Elev= 30
  4648.5  474.29  4707.1  474.34  4817.8  471.57  4828.1  472.21  4891.9  469.33
  4939.4  466.92  4949.5  465.24  4955.8  462.23  4960.9  460.82  4969.7  457.23
  4979.8  455.59  4989.9  452.65  5009.9  449.89  5013.2  450.39  5030.4  460.48
  5050.6  461.12  5101.2  459.58  5131.5  459.75  5182.1  461.99  5202.3  461.55
  5242.8  463.02  5310.7  461.95  5428.6  461.32  5581.3  462.92  5743.4  463.83
  5914.6  466.17  5973.1  467.88  6158.9  475.57  6409.3  488.85  6544.8  493.24
#Mann= 6 ,-1 , 0
  4648.5      .1       0  4707.1     .16       0  4955.8     .07       0
  5182.1     .12       0  5310.7      .1       0  5581.3     .05       0
Bank Sta=4960.9,5030.4
XS Rating Curve= 0 ,0
Exp/Cntr=0.3,0.1

Type RM Length L Ch R = 1 ,68290   ,350,350,350
BEGIN DESCRIPTION:
PLUMMERS CREEK 57.0
END DESCRIPTION:
XS GIS Cut Line= 5
      3493057.31     10583847.72      3492974.84     10583292.14
      3492710.09     10583192.31      3492380.23     10583231.37
       3491451.4     10582931.89
#Sta/Elev= 30
  4270.9   469.4  4378.1  469.42    4406  468.29  4469.1  468.08  4539.8  465.72
  4614.3  464.76  4812.5  458.26    4880  457.68  4953.1  459.33  4965.3  456.28
  4974.4  451.53  4989.9  448.33  5006.5  449.49    5015  453.45  5038.6  456.25
  5081.3  459.27  5115.5  460.13  5150.5  456.05  5155.6  457.14  5173.9  456.94
  5181.1  458.31    5194  459.44  5224.3  458.64  5288.7  459.26  5480.7  461.59
  5582.3  462.67  5985.7  470.81  6151.2  476.31  6317.8  483.91  6423.6  487.33
#Mann= 6 ,-1 , 0
  4270.9     .05       0  4953.1    .035       0  5081.3      .1       0
  5181.1     .16       0  5288.7      .1       0  5480.7     .05       0
Bank Sta=4965.3,5038.6
XS Rating Curve= 0 ,0
Exp/Cntr=0.3,0.1

Type RM Length L Ch R = 1 ,67940   ,427,427,427
BEGIN DESCRIPTION:
PLUMMERS CREEK 56.0
END DESCRIPTION:
XS GIS Cut Line= 4
      3493074.67     10583695.81      3493083.35     10583391.96
      3492601.58     10582693.18      3492163.19     10581959.63
#Sta/Elev= 30
  4185.9  468.32  4220.1  468.64  4380.1  463.21  4612.2     458  4671.7  457.53
  4728.5  459.35  4800.2  458.27  4821.1  459.45  4943.5  457.54  4958.4  455.47
  4994.2  449.06  5000.2  446.78  5015.2  449.44    5024  454.82  5036.8  458.96
  5182.2  463.41  5215.1  462.42    5260  463.67  5274.9  465.33  5362.4  467.13
  5398.7  466.52  5463.5  469.49  5521.9  470.56  5564.7  469.29    5612  472.08
  5619.2  472.22  5801.8  474.67  5887.6  478.06  5988.8  482.38  6193.2  488.24
#Mann= 8 ,-1 , 0
  4185.9     .05       0  4943.5     .07       0  5036.8      .1       0
  5215.1     .05       0    5612      .1       0  5619.2     .05       0
  5801.8      .1       0  5887.6     .05       0
Bank Sta=4958.4,5024
XS Rating Curve= 0 ,0
Exp/Cntr=0.3,0.1

Type RM Length L Ch R = 1 ,67513   ,280,280,280
BEGIN DESCRIPTION:
PLUMMERS CREEK 55.5
END DESCRIPTION:
XS GIS Cut Line= 4
      3493278.66      10583782.6       3493217.9      10583266.1
       3493174.5     10582758.28      3492822.95     10582176.71
#Sta/Elev= 30
  4182.3  467.56  4253.7  464.54  4445.1     461  4847.3  457.37  4887.5  458.12
  4927.6  457.05  4944.6  457.85  4949.6  455.95  4957.7  456.17 4961.29  453.78
  4967.8   448.3  4977.6  445.17  4997.9   446.1  5007.9  447.62    5018  450.69
  5068.6  453.39  5088.2  453.13  5098.3  451.48  5158.5  454.07    5212  453.58
  5219.8   454.6    5226  458.18  5241.5  459.16  5363.7  462.17  5553.9  472.66
  5691.6  477.99  5728.5  480.55  5749.9  480.55  5786.7  484.35  5891.6  491.66
#Mann= 3 , 0 , 0
  4182.3     .05       0 4961.29    .035       0  5068.6     .05       0
Bank Sta=4961.29,5068.6
XS Rating Curve= 0 ,0
Exp/Cntr=0.3,0.1

Type RM Length L Ch R = 1 ,67233   ,245,245,245
BEGIN DESCRIPTION:
PLUMMERS CREEK 55.0
END DESCRIPTION:
XS GIS Cut Line= 4
      3493387.17     10583782.57      3493313.38     10583070.78
      3493413.21     10582806.03      3492936.47     10582203.59
#Sta/Elev= 30
  4093.3  466.74  4124.4  466.25  4144.5  467.35  4335.5  461.03  4784.6  457.55
  4833.3  457.39    4907  458.06  4925.5  456.85 4930.03  455.03  4937.2  452.81
    4979  450.65  4992.3  445.93  5000.1  445.22    5011   448.3  5017.1  454.12
  5022.5  455.17    5042  457.74  5072.2  460.33  5165.7  461.35  5175.5  462.04
  5216.5  463.13    5231   462.1  5295.1  462.33  5458.5  466.69  5650.9  475.98
  5671.7  478.52    5715  479.05  5729.4  480.81  5750.2  480.26  5860.1  488.01
#Mann= 7 ,-1 , 0
  4093.3     .05       0  4784.6     .16       0  4833.3     .05       0
    4907    .035       0    5042     .05       0  5165.7     .08       0
  5175.5     .05       0
Bank Sta=4930.03,5022.5
XS Rating Curve= 0 ,0
Exp/Cntr=0.3,0.1

Type RM Length L Ch R = 1 ,66988   ,398,398,398
BEGIN DESCRIPTION:
PLUMMERS CREEK 54.0
END DESCRIPTION:
XS GIS Cut Line= 4
      3493560.78     10584407.62       3493552.1     10583183.63
       3493595.5     10582905.85      3493322.77     10582234.83
#Sta/Elev= 30
  3608.7  470.94  3994.7   464.8  4214.7  463.78  4484.7  459.74  4524.7  459.88
  4544.7  461.02  4604.7  459.24  4764.7  457.19  4824.7  458.64  4860.9  457.72
  4885.3  457.75  4915.7   456.2  4925.3  455.04  4930.4  453.05  4956.2  454.47
  4966.3  453.49  4986.6  448.64    4998  444.51  5006.8  445.43    5027  453.82
  5047.3  455.74  5135.4  457.43  5217.8  458.32    5433   462.3  5474.6  463.01
  5563.7  466.77  5696.4  474.22  5707.5   475.1  5815.1  481.23  5838.2  482.35
#Mann= 9 ,-1 , 0
  3608.7     .05       0  4860.9     .16       0  4885.3     .07       0
  5135.4     .16       0  5217.8     .08       0    5433     .05       0
  5696.4     .08       0  5707.5     .05       0  5815.1      .1       0
Bank Sta=4966.3,5027
XS Rating Curve= 0 ,0
Exp/Cntr=0.3,0.1

Type RM Length L Ch R = 1 ,66590   ,1246,1246,1246
BEGIN DESCRIPTION:
PLUMMERS CREEK 53.0
END DESCRIPTION:
XS GIS Cut Line= 4
      3493799.49     10584233.93      3493764.77     10583439.71
      3493912.34     10582654.12      3493322.04     10582059.47
#Sta/Elev= 30
    3704  470.45  3984.6  466.32  4032.8  466.65  4196.8  463.88  4326.9  464.27
  4564.5  457.59  4640.6  456.37  4700.5  456.38  4771.7  454.63  4802.3  456.07
  4812.4  455.62  4832.2     452  4934.5  453.42  4975.2   449.4  4999.6  443.05
  5002.9  443.55  5026.1  452.75  5036.3  455.25  5046.5  456.03  5066.8  454.96
    5077   452.3  5104.9  454.95  5152.8  457.14  5400.8  462.35  5537.1  464.98
  5618.4  467.13  5766.9  473.72  5883.1  477.36  6021.5  482.44  6136.2  485.09
#Mann= 9 ,-1 , 0
    3704      .1       0  4032.8     .05       0  4640.6     .16       0
  4812.4     .07       0  5046.5     .12       0  5152.8     .16       0
  5400.8     .12       0  5537.1     .16       0  5883.1     .05       0
Bank Sta=4934.5,5026.1
XS Rating Curve= 0 ,0
Exp/Cntr=0.3,0.1
