--- BUCK CREEK.prj (project) ---

Proj Title=BUCK CREEK Base Level Engineering
Current Plan=p01
Default Exp/Contr=0.3,0.1
English Units
Geom File=g01
Flow File=f01
Plan File=p01
Y Axis Title=Elevation
X Axis Title(PF)=Main Channel Distance
X Axis Title(XS)=Station
BEGIN DESCRIPTION:
BUCK CREEK
END DESCRIPTION:
DSS Export Rating Curves= 0
DSS Export Rating Curve Sorted= 0
DSS Export Volume Flow Curves= 0
DXF OffsetX= 0
DXF OffsetY= 0
DXF ScaleX= 1
DXF ScaleY= 10

--- BUCK CREEK.p01 (plan) ---

Plan Title=Multiple Run
Short Identifier=Multiple
Geom File=g01
Flow File=f01
Subcritical Flow
K Sum by GR= 0
Std Step Tol= 0.01
Critical Tol= 0.01
Num of Std Step Trials= 20
Max Error Tol= 0.3
Flow Tol Ratio= 0.001
Split Flow NTrial= 30
Split Flow Tol= 0.02
Split Flow Ratio= 0.02
Log Output Level= 0
Friction Slope Method= 1
Unsteady Friction Slope Method= 2
Unsteady Bridges Friction Slope Method= 1
Parabolic Critical Depth
Global Vel Dist=  1 , 1 , 1
Global Log Level= 0
CheckData=True
Encroach Param= -1, 0, 0, 0
BEGIN DESCRIPTION:
Multiple Run
END DESCRIPTION:

--- BUCK CREEK.f01 (steady flow) ---

Flow Title=Multiple
Program Version=4.10
Number of Profiles= 7
Profile Names=10-year,25-year,50-year,1pct_min,100-year,1pct_plu,500-year
River Rch & RM=BUCK CREEK,Reach-1         ,28797
    1940    2774    3489    3198    4325    5849    6629
River Rch & RM=BUCK CREEK,Reach-1         ,21186
    2462    3560    4512    4162    5628    7612    8741
River Rch & RM=BUCK CREEK,Reach-1         ,17349
    2562    3706    4698    4333    5860    7926    9101
River Rch & RM=BUCK CREEK,Reach-1         ,16343
    4491    6646    8554    7999   10818   14630   17266
River Rch & RM=BUCK CREEK,Reach-1         ,11802
    5412    8049   10394    9743   13177   17820   21139
River Rch & RM=BUCK CREEK,Reach-1         ,10973
    5412    8049   10394    9743   13177   17820   21139
River Rch & RM=BUCK CREEK,Reach-1         ,5432
    5418    8040   10365    9700   13118   17741   20972
Boundary for River Rch & Prof#=BUCK CREEK,Reach-1         , 1
Up Type= 0
Dn Type= 3
Dn Slope=0.004
Boundary for River Rch & Prof#=BUCK CREEK,Reach-1         , 2
Up Type= 0
Dn Type= 3
Dn Slope=0.004
Boundary for River Rch & Prof#=BUCK CREEK,Reach-1         , 3
Up Type= 0
Dn Type= 3
Dn Slope=0.004
Boundary for River Rch & Prof#=BUCK CREEK,Reach-1         , 4
Up Type= 0
Dn Type= 3
Dn Slope=0.004
Boundary for River Rch & Prof#=BUCK CREEK,Reach-1         , 5
Up Type= 0
Dn Type= 3
Dn Slope=0.004
Boundary for River Rch & Prof#=BUCK CREEK,Reach-1         , 6
Up Type= 0
Dn Type= 3
Dn Slope=0.004
Boundary for River Rch & Prof#=BUCK CREEK,Reach-1         , 7
Up Type= 0
Dn Type= 3
Dn Slope=0.004
DSS Import GetInterval= 0
DSS Import GetPeak= 0
DSS Import FillOption= 0

--- BUCK CREEK.g01 (geometry) ---

Geom Title=Existing Conditions
Program Version=4.10

River Reach=BUCK CREEK      ,Reach-1
Reach XY= 30
      3607552.11     10442361.64      3606992.37     10442062.84
      3605843.65     10442078.03      3605048.54     10441657.42
      3603211.98     10442640.72      3602626.14     10442244.08
      3601639.38     10442357.67      3600606.62     10441613.28
      3599017.07     10441621.33      3598756.52     10441393.72
      3597547.91     10441263.49      3596899.56     10441705.05
      3596822.28      10442181.3      3595742.43     10442911.57
      3595546.64     10443462.21      3595117.41     10443684.79
      3594524.69     10444866.23      3593903.57     10444965.19
      3593298.94     10445425.37      3592266.36     10445719.85
      3592021.62       10445471.      3591079.81     10445563.26
      3590710.97     10445425.59      3590350.49     10445581.05
      3590355.04     10446101.86      3589416.86     10446899.61
      3588381.59     10446212.62      3587013.47     10446565.18
       3586930.8     10447784.26      3586702.11     10447921.64

Type RM Length L Ch R = 1 ,28797   ,641,641,641
BEGIN DESCRIPTION:
UNT0277 IN DUCK CR 5 0
END DESCRIPTION:
XS GIS Cut Line= 2
      3607652.34     10441792.38      3607397.13     10442891.33
#Sta/Elev= 30
  4405.6  489.79  4429.6  489.08  4472.3  489.61  4514.9  488.63    4520   487.8
  4548.6  488.23  4605.3   486.8  4610.4  485.73  4647.9  485.54  4743.6  478.49
  4907.9  468.32  4961.8  462.93  4979.7  453.89    4990  447.15    4997  443.69
  4997.3  443.19  5001.6  443.69  5004.4  443.85  5010.5  447.41  5020.8  456.57
 5027.74  464.94  5031.1  467.73  5047.1  474.17  5052.2  473.61  5072.1  476.92
  5180.1  485.89  5369.9   496.8  5431.5  498.67  5488.8  501.59  5533.8  502.49
#Mann= 3 ,-1 , 0
  4405.6     .16       0    4997     .07       0  5001.6     .16       0
Bank Sta=4961.8,5027.74
XS Rating Curve= 0 ,0
Exp/Cntr=0.3,0.1

Type RM Length L Ch R = 1 ,28156   ,776,776,776
BEGIN DESCRIPTION:
UNT0277 IN DUCK CR 4 0
END DESCRIPTION:
XS GIS Cut Line= 3
      3607162.77     10441693.38      3607058.59     10441922.57
      3606985.72     10442797.08
#Sta/Elev= 30
  4568.6  490.12  4611.3  488.97    4675  489.63  4742.4  487.21  4822.4  477.97
  4869.6  470.49  4909.7     467  4929.8  459.87  4949.9  456.94  4969.9   451.2
    4990  442.77  4997.7  442.04  4998.1  441.54  5002.4  442.04  5010.1  448.15
  5030.2  459.52  5040.2  462.77  5070.3  463.82  5077.2  463.22  5082.2  459.18
  5090.4  459.45  5110.4  464.58  5120.5  466.04  5170.6  468.09  5197.6  470.72
  5220.8  470.94  5301.1  474.73  5380.8  480.91  5501.8  489.08  5697.9  496.77
#Mann= 4 ,-1 , 0
  4568.6     .16       0  4997.7     .07       0  5002.4     .16       0
  5380.8      .1       0
#XS Ineff= 2 , 0
                         5068.46          463.88
Permanent Ineff=
       F       F
Bank Sta=4949.9,5030.2
XS Rating Curve= 0 ,0
Exp/Cntr=0.3,0.1

Type RM Length L Ch R = 1 ,27380   ,779,779,779
BEGIN DESCRIPTION:
UNT0277 IN DUCK CR 37 0
END DESCRIPTION:
XS GIS Cut Line= 4
      3606350.26     10441610.12       3606313.8     10441932.99
       3606313.8     10442255.91      3606584.63     10442844.44
#Sta/Elev= 30
  4538.3  477.78  4590.2  476.81  4640.5   472.1  4655.5  472.16  4700.9  468.03
  4745.4   466.2  4871.9  457.29  4961.9  455.87  4971.9  453.86 4977.07  450.17
  4999.5  435.81  4999.8  435.31  5004.3  435.81  5021.9  443.15  5051.9  449.78
  5061.9   450.5  5071.9  449.74  5081.9  447.11  5091.9  447.45  5151.9  457.15
  5161.9  455.47  5181.5   457.7    5196  456.73  5203.5  459.53  5241.9  460.98
  5310.8  466.68  5362.3  468.36    5603  483.65  5700.4  488.61    5834  492.16
#Mann= 3 ,-1 , 0
  4538.3     .16       0  4999.5     .07       0  5004.3     .16       0
Bank Sta=4977.07,5051.9
XS Rating Curve= 0 ,0
Exp/Cntr=0.3,0.1

Type RM Length L Ch R = 1 ,26601   ,773,773,773
BEGIN DESCRIPTION:
UNT0277 IN DUCK CR 36 0
END DESCRIPTION:
XS GIS Cut Line= 4
      3606016.94     10441115.25      3605766.93     10441776.74
      3605584.63     10442037.16      3605569.01     10442896.58
#Sta/Elev= 30
  4169.2  498.49  4260.8  489.81  4450.1   468.2  4603.6  457.48  4620.5  452.85
  4650.7  455.68  4665.8  449.48  4675.5  443.45  4689.2  445.53  4705.7  453.11
    4711  450.32  4730.5   453.6  4838.1  452.38  4926.7  450.48  4932.8  446.21
  4947.6  437.78  4968.6  435.89  4980.8  430.42  4981.2  429.92  4985.9  430.42
    5013  432.02  5063.6  446.66  5077.6  452.02  5119.2  452.99  5316.6   462.7
  5414.7  471.98  5512.7  475.61  5613.6  478.37  5706.9  479.64  6053.8  483.19
#Mann= 12 ,-1 , 0
  4169.2     .05       0  4260.8     .16       0  4665.8      .1       0
  4838.1     .16       0  4980.8     .07       0  4985.9     .16       0
  5119.2      .1       0  5316.6     .05       0  5414.7      .1       0
  5512.7     .05       0  5613.6      .1       0  5706.9     .05       0
#XS Ineff= 2 , 0
         4773.84  453.79
Permanent Ineff=
       F       F
Bank Sta=4932.8,5063.6
XS Rating Curve= 0 ,0
Exp/Cntr=0.3,0.1

Type RM Length L Ch R = 1 ,25828   ,611,611,611
BEGIN DESCRIPTION:
UNT0277 IN DUCK CR 34 0
END DESCRIPTION:
XS GIS Cut Line= 4
      3605417.99      10440714.2      3605048.18     10441479.86
      3605037.76     10441953.82      3605360.67      10442891.3
#Sta/Elev= 30
  3971.4  502.94  4137.5  488.36  4154.6  489.19  4373.8  476.29  4501.3  471.91
  4606.5  466.17  4730.7  453.91  4798.5  449.38    4923  446.76  4933.5  445.27
  4953.5  439.39  4963.5  440.23  4983.5   427.9  5000.8  424.46  5001.2  423.96
  5006.3  424.46  5043.5  443.83  5063.5  446.21  5273.6   446.7  5388.1   451.5
  5493.4  456.37  5598.6  463.92  5665.6  466.02  5691.5  462.94  5716.5  463.22
    5809  470.11  6003.7  478.27  6234.8  484.82  6266.5  488.02  6287.3  486.39
#Mann= 11 ,-1 , 0
  3971.4     .16       0  4373.8      .1       0  4501.3     .16       0
  4606.5      .1       0    4923     .16       0  5000.8     .07       0
  5006.3     .16       0  5388.1      .1       0  5493.4     .05       0
  5598.6     .16       0    5809     .05       0
Bank Sta=4933.5,5043.5
XS Rating Curve= 0 ,0
Exp/Cntr=0.3,0.1

Type RM Length L Ch R = 1 ,25217   ,954,954,954
BEGIN DESCRIPTION:
UNT0277 IN DUCK CR 30 0
END DESCRIPTION:
XS GIS Cut Line= 4
      3604272.12     10441057.96      3604647.13     10441719.45
      3604662.76     10442235.07      3605021.95     10442917.01
#Sta/Elev= 30
  4006.9  498.07  4113.6  492.52  4335.5  474.75  4470.9  462.88  4549.2  458.26
  4646.4  450.87  4700.8  446.76  4839.5  442.58  4869.5  433.92  4889.5  441.26
  4939.6  442.73  4959.6  441.02  4979.6  431.53    4997  419.02  5002.1  419.02
  5019.6  433.92  5029.6   439.8  5049.6  443.56  5149.7  446.76  5332.8  457.97
  5376.8  458.18  5465.4  462.92  5613.5  468.26  5720.6  468.67  5762.1  468.96
  5767.7  466.95  5789.8  465.82  5844.4   471.5  5956.5  475.86  6053.9  479.55
#Mann= 9 ,-1 , 0
  4006.9     .16       0  4335.5      .1       0  4549.2     .05       0
  4646.4     .16       0  4979.6     .07       0  5019.6     .16       0
  5465.4      .1       0  5720.6     .16       0  5956.5     .05       0
#XS Ineff= 2 , 0
          4938.6  442.53
Permanent Ineff=
       F       F
Bank Sta=4979.6,5019.6
XS Rating Curve= 0 ,0
Exp/Cntr=0.3,0.1

Type RM Length L Ch R = 1 ,24263   ,698,698,698
BEGIN DESCRIPTION:
UNT0277 IN DUCK CR 3 0
END DESCRIPTION:
XS GIS Cut Line= 3
      3603891.93     10441313.25      3603959.63     10442110.07
      3604344.85     10443047.08
#Sta/Elev= 30
  4037.4  510.16  4333.3  471.53  4566.8  449.89  4685.8  442.39  4822.8  437.87
  4934.4  437.19  4962.5  436.13  4968.5  432.43  4986.5  416.65  4997.9  414.55
  4998.4  414.05  5004.1  414.55  5039.8  431.77  5069.2  437.26  5076.7  431.82
  5087.5  430.66  5093.2  436.14  5098.6  432.54  5117.1  438.53  5122.5  435.68
  5141.1  439.04  5146.5  436.19  5170.5  439.89  5175.9  436.91  5194.4   437.7
  5199.8  433.59  5210.8  435.03  5684.3  456.84  5685.4  456.87  5850.2  464.02
#Mann= 9 ,-1 , 0
  4037.4     .16       0  4685.8      .1       0  4822.8     .16       0
  4934.4     .05       0  4997.9     .04       0  5004.1     .05       0
  5210.8     .16       0  5684.3     .05       0  5685.4     .16       0
Bank Sta=4968.5,5039.8
XS Rating Curve= 0 ,0
Exp/Cntr=0.3,0.1

Type RM Length L Ch R = 1 ,23565   ,867,867,867
BEGIN DESCRIPTION:
UNT0277 IN DUCK CR 29 0
END DESCRIPTION:
XS GIS Cut Line= 3
      3603371.09     10441130.94      3603350.26     10442401.74
      3603818.06     10443222.98
#Sta/Elev= 30
  3595.7  533.07  3616.4  530.02  3676.4  515.32  3716.4  502.99  3736.4  498.96
  3916.4  480.66  4036.5   471.1  4156.5  458.67  4216.5  453.82  4445.3  438.21
  4496.5  435.85  4676.5  433.67  4716.6  432.19  4903.8  432.65  4962.8  432.09
  4970.1  430.76  4984.5   421.2  4997.1  411.26  4997.6  410.76  5003.5  411.26
  5016.2  417.27  5027.7  425.34  5037.8  429.89  5043.5  427.19  5050.7  431.05
  5065.1  433.07  5279.8     442  5506.1  454.02  5633.8  455.89  5811.8  458.34
#Mann= 4 ,-1 , 0
  3595.7     .16       0  4997.1     .07       0  5003.5     .16       0
  5633.8     .05       0
Bank Sta=4970.1,5037.8
XS Rating Curve= 0 ,0
Exp/Cntr=0.3,0.1

Type RM Length L Ch R = 1 ,22698   ,741,741,741
BEGIN DESCRIPTION:
UNT0277 IN DUCK CR 27 0
END DESCRIPTION:
XS GIS Cut Line= 4
      3603121.09     10441073.66      3602963.46     10442320.84
      3602834.63     10442599.66      3603141.95     10443130.94
#Sta/Elev= 30
  3646.7  533.06  3754.3  506.39  3785.8  500.31  3834.5  493.78  3994.9  479.14
  4160.4  466.24    4199  461.76  4269.6  459.47  4672.8  433.62    4943  428.93
  4959.8  420.84  4971.5  414.02  4981.8  412.43  4994.4  407.17  5000.5  406.94
    5001  406.44  5007.1  406.94  5011.8  408.64  5025.9  419.99  5034.8  426.44
  5047.9  429.14    5132  431.25  5206.3  429.64  5270.5  430.77  5490.1  437.42
  5538.9  440.21    5592  440.16  5619.3  442.24  5731.2  444.72  5824.7  450.51
#Mann= 3 ,-1 , 0
  3646.7     .16       0  5000.5     .07       0  5007.1     .16       0
Bank Sta=4959.8,5025.9
XS Rating Curve= 0 ,0
Exp/Cntr=0.3,0.1

Type RM Length L Ch R = 1 ,21957   ,771,771,771
BEGIN DESCRIPTION:
UNT0277 IN DUCK CR 25 0
END DESCRIPTION:
XS GIS Cut Line= 3
      3602324.22     10440844.47      3602308.59     10442224.66
      3602506.26     10443207.81
#Sta/Elev= 30
  3517.1  503.62  3954.3  466.66  4064.3  459.89  4264.3  452.49  4284.3  449.49
  4514.3  457.13  4734.3  449.45  4945.5   430.1  4955.5  428.65  4965.7  421.02
    4993  404.04  4993.5  403.54  4999.6  404.04  5042.1  417.05  5057.5  410.85
  5077.9  407.35  5087.9   406.2    5093  413.44  5108.5  407.21  5138.3  405.78
  5143.8  409.52  5179.9  405.74  5240.5  417.73  5251.3  424.06  5403.3   432.6
  5550.5  435.63  5707.5  442.16  5808.4  446.71  5834.9  447.47  5900.2  450.59
#Mann= 9 ,-1 , 0
  3517.1     .16       0    4993     .07       0  4999.6     .16       0
  5138.3      .1       0  5403.3     .05       0  5550.5      .1       0
  5707.5     .05       0  5808.4      .1       0  5834.9     .05       0
Bank Sta=4965.7,5042.1
XS Rating Curve= 0 ,0
Exp/Cntr=0.3,0.1

Type RM Length L Ch R = 1 ,21186   ,785,785,785
BEGIN DESCRIPTION:
UNT0277 IN DUCK CR 24 0
END DESCRIPTION:
XS GIS Cut Line= 4
      3602188.81     10440787.12      3601678.38     10442261.11
      3601605.47     10442516.32      3601459.65     10442932.95
#Sta/Elev= 30
  3336.5  499.51  3375.3  495.38  3595.3  479.44  3712.7  473.68  3849.2  470.46
  4107.1  459.23  4219.6  452.12    4339  440.93  4420.7  435.39  4484.2  432.41
  4815.2  423.23  4844.2  421.96  4886.3  422.11  4928.1  419.27  4948.9  410.07
  4959.3  407.21  4974.4  405.74    4997  401.39  4997.5  400.89  5004.9  401.39
  5008.2  405.01  5013.4  405.93  5021.8  415.46  5032.1  420.24  5047.2  421.36
  5114.8  421.81  5209.8  424.66  5278.3  428.56  5495.9  445.35  5603.2  448.37
#Mann= 6 ,-1 , 0
  3336.5     .16       0    4339     .05       0  4815.2     .16       0
    4997     .07       0  5004.9     .16       0  5021.8     .05       0
Bank Sta=4928.1,5032.1
XS Rating Curve= 0 ,0
Exp/Cntr=0.3,0.1

Type RM Length L Ch R = 1 ,20401   ,772,772,772
BEGIN DESCRIPTION:
UNT0277 IN DUCK CR 2 1
END DESCRIPTION:
XS GIS Cut Line= 2
      3601865.86     10440594.49      3600803.97      10442447.6
#Sta/Elev= 30
  3332.3  494.13    3515  477.56  3611.4  470.47  3743.9  464.61  3912.1  453.09
  4132.2  440.57  4389.4  430.35    4447  426.66  4489.7  426.61  4600.3  421.12
  4717.7   416.3  4824.6   415.6  4937.8  414.83  4959.4  409.64  4975.2  407.73
  4996.8  397.58  5007.7  397.36  5008.2  396.86  5015.8  397.36  5018.4  399.91
    5040  406.31  5055.8  416.97  5069.4  423.49  5104.7  427.51  5179.5   432.1
  5185.3   433.9  5374.7  433.24  5389.2  432.51    5427  430.29  5468.1   432.8
#Mann= 8 ,-1 , 0
  3332.3     .16       0  4489.7      .1       0  4600.3     .05       0
  4824.6     .16       0  5007.7     .07       0  5015.8     .16       0
  5374.7      .1       0  5389.2     .05       0
Bank Sta=4937.8,5055.8
XS Rating Curve= 0 ,0
Exp/Cntr=0.3,0.1

Type RM Length L Ch R = 1 ,19629   ,855,855,855
BEGIN DESCRIPTION:
UNT0277 IN DUCK CR 2 0
END DESCRIPTION:
XS GIS Cut Line= 4
      3600647.13     10440339.27      3600459.63     10441516.32
      3600464.84     10441781.95      3600652.24     10442417.01
#Sta/Elev= 30
  3702.7  453.01  3748.1  450.54  3768.7  449.83  3867.1   442.2  4067.3  433.84
  4253.3  430.45  4292.4  428.43  4515.2  421.83  4687.3   414.2  4900.1  410.84
  4959.9  410.95  4969.9  407.71  4989.9   396.4  4995.7  395.46  4996.2  394.96
  5004.1  395.46  5009.9  395.91  5019.9  404.59  5039.9  411.98  5064.7  414.45
  5166.7  420.38  5343.7  426.71  5592.4   432.4  5608.3  436.09  5639.6  432.27
  5659.1  433.61  5664.3  431.78  5670.8  433.41  5681.3  433.95  5822.4  435.07
#Mann= 8 ,-1 , 0
  3702.7     .16       0  3748.1     .05       0  4067.3     .16       0
  4253.3     .05       0  4900.1     .16       0  4995.7     .07       0
  5004.1     .16       0  5064.7     .05       0
Bank Sta=4959.9,5039.9
XS Rating Curve= 0 ,0
Exp/Cntr=0.3,0.1

Type RM Length L Ch R = 1 ,18774   ,578,578,578
BEGIN DESCRIPTION:
UNT0277 IN DUCK CR 19 0
END DESCRIPTION:
XS GIS Cut Line= 3
      3599742.28     10440817.53      3599697.14     10441827.96
      3599971.44      10442373.1
#Sta/Elev= 30
    4155  419.78  4267.6  419.05  4299.3  419.51  4429.4   412.5  4520.6  408.85
  4609.6  405.34  4649.6   404.5  4739.7  405.81  4757.7  405.39  4839.8  405.38
  4889.8  403.84    4934  405.15  4959.9  405.39    4973  404.63  4979.9  403.51
  4989.9  395.55  4995.4   393.2  4995.9   392.7  5004.5   393.2    5010  393.42
    5020  397.77    5030  404.06    5040  405.99  5056.6  406.02  5232.6  406.26
  5383.2  407.56  5478.1   413.7  5567.4  417.21  5685.5  419.98  5776.7  420.05
#Mann= 8 ,-1 , 0
    4155     .05       0  4520.6     .16       0  4757.7     .05       0
    4934     .16       0    4973      .1       0  4995.4     .07       0
  5004.5      .1       0  5056.6     .05       0
#XS Ineff= 2 , 0
         4937.43   405.6
Permanent Ineff=
       F       F
Bank Sta=4973,5040
XS Rating Curve= 0 ,0
Exp/Cntr=0.3,0.1

Type RM Length L Ch R = 1 ,18196   ,847,847,847
BEGIN DESCRIPTION:
UNT0277 IN DUCK CR 17 0
END DESCRIPTION:
XS GIS Cut Line= 3
      3599092.11     10441141.65      3599142.11     10441591.64
       3599392.1     10442391.63
#Sta/Elev= 30
  4547.5   411.5  4658.2  408.34  4829.2  401.39  4859.4  398.83  4879.5     394
  4889.6  393.39  4909.7  400.57  4970.1  401.04  4980.1  397.35  4985.6  392.51
  4986.1  392.01  4994.7  392.51  5002.9  392.93  5016.5  396.71  5021.7  396.49
    5049  401.05  5063.1  401.04  5086.7  399.04  5094.6  399.04  5151.7  400.01
  5174.7  401.35  5189.4  401.96  5319.3  402.53  5351.8  401.41  5384.2  401.35
  5440.3  402.32  5534.6  405.34  5616.8  410.97  5724.7  421.07  5838.4   427.8
#Mann= 4 ,-1 , 0
  4547.5     .16       0  4985.6     .07       0  4994.7     .16       0
  5174.7     .05       0
Bank Sta=4970.1,5049
XS Rating Curve= 0 ,0
Exp/Cntr=0.3,0.1

Type RM Length L Ch R = 1 ,17349   ,523,523,523
BEGIN DESCRIPTION:
UNT0277 IN DUCK CR 16 0
END DESCRIPTION:
XS GIS Cut Line= 4
      3598470.05     10441068.44      3598423.18     10441354.86
      3598407.55     10441636.11      3598192.11     10442091.62
#Sta/Elev= 30
  4612.6  422.72  4630.9  422.46  4692.3  416.39  4697.4  416.58  4753.6  412.16
  4758.7  412.37  4788.1  409.94    4815  406.54  4820.1  406.85  4876.4  402.12
  4949.7  397.61  4989.7  393.26  4994.9  390.67  4995.4  390.17  5004.6  390.67
  5013.5  391.89  5019.8  396.44  5029.8  398.02  5034.1  397.84  5069.9  397.13
  5132.2  397.69  5230.8  398.58  5389.7   403.2  5509.4  410.76    5515  410.56
  5588.9  416.15    5622  417.54  5644.2  419.73  5666.3  422.93  5688.4  423.56
#Mann= 5 ,-1 , 0
  4612.6     .16       0  4994.9     .07       0  5004.6     .16       0
  5034.1      .1       0  5132.2     .05       0
Bank Sta=4949.7,5029.8
XS Rating Curve= 0 ,0
Exp/Cntr=0.3,0.1

Type RM Length L Ch R = 1 ,16826   ,483,483,483
BEGIN DESCRIPTION:
UNT0277 IN DUCK CR 14 0
END DESCRIPTION:
XS GIS Cut Line= 3
      3598326.52     10440940.06      3597968.41     10441141.91
      3597777.42     10441823.37
#Sta/Elev= 30
  4406.7  424.35  4462.1  424.04  4518.7  421.87  4564.7  420.64  4634.7  420.87
  4698.7  419.11  4750.8  412.96  4791.5  407.67  4820.2  405.68  4838.3  403.15
  4856.8     402  4861.9  400.81  4888.7  399.53  4930.2  395.86  4974.7  396.84
  4983.7  394.86  4989.2   388.4  4989.7   387.9    4999   388.4  5008.8   389.9
  5014.8  393.02  5042.9  395.78  5052.3  395.64  5108.3  396.15  5222.5  400.66
  5295.2  404.99    5316  407.65  5409.5  414.29  5420.3  415.95  5525.5  420.26
#Mann= 8 ,-1 , 0
  4406.7     .16       0  4518.7     .05       0  4634.7     .16       0
  4750.8      .1       0  4888.7     .16       0  4989.2     .07       0
    4999     .16       0  5052.3     .05       0
Bank Sta=4983.7,5014.8
XS Rating Curve= 0 ,0
Exp/Cntr=0.3,0.1

Type RM Length L Ch R = 1 ,16343   ,411,411,411
BEGIN DESCRIPTION:
UNT0277 IN DUCK CR 13 0
END DESCRIPTION:
XS GIS Cut Line= 3
      3597122.07     10440712.25       3597321.7      10441055.1
      3597737.75     10441802.69
#Sta/Elev= 30
  4295.8  416.79  4362.1  415.09  4367.9   415.6  4501.1  408.95  4624.3  405.38
  4726.4  400.02  4860.2  396.39  4913.1  395.86  4948.2  394.82    4986  390.28
  4991.7  386.91  4992.2  386.41  5003.4  386.91  5007.7  387.26  5035.2  394.78
  5051.2   395.3  5101.8  394.37  5169.2  396.33  5197.5  398.31  5261.2   404.7
  5294.7   408.1  5300.4  407.59  5338.2  412.41  5365.6   413.6  5381.6  415.55
  5425.1  416.56  5441.1  418.68  5446.8  418.08  5481.5  419.24  5548.1   420.2
#Mann= 7 ,-1 , 0
  4295.8      .1       0  4913.1     .16       0  4991.7     .07       0
  5003.4     .16       0  5101.8     .05       0  5261.2      .1       0
  5481.5     .05       0
Bank Sta=4948.2,5035.2
XS Rating Curve= 0 ,0
Exp/Cntr=0.3,0.1

Type RM Length L Ch R = 1 ,15932   ,535,535,535
BEGIN DESCRIPTION:
UNT0277 IN DUCK CR 10 0
END DESCRIPTION:
XS GIS Cut Line= 3
      3596942.11     10441041.67      3597142.11     10441541.64
      3597592.07     10441741.63
#Sta/Elev= 30
  4461.8  420.38  4494.1   420.3    4624  407.15    4731  399.01  4811.1  395.91
    4902  394.35  4914.1  393.95  4931.6  391.84    4937  392.52  4946.4  390.06
  4978.8  389.67  4985.5  386.87  4990.9  386.95  4991.7  385.75  4992.2  385.25
  5003.4  385.75  5009.2  385.86  5014.7  390.56  5022.2  389.48  5032.4  389.51
  5037.9  392.47  5089.9  394.87  5153.5  393.42  5197.3  393.38  5273.2  396.99
  5295.7  398.61  5339.5  402.96  5356.6  405.66    5438  413.44  5492.7  416.96
#Mann= 7 ,-1 , 0
  4461.8     .16       0    4624      .1       0  4811.1     .16       0
  4991.7     .07       0  5003.4     .16       0  5273.2     .05       0
  5295.7      .1       0
Bank Sta=4937,5037.9
XS Rating Curve= 0 ,0
Exp/Cntr=0.3,0.1

Type RM Length L Ch R = 1 ,15397   ,872,872,872
BEGIN DESCRIPTION:
UNT0277 IN DUCK CR 21 1
END DESCRIPTION:
XS GIS Cut Line= 4
      3596298.28     10441360.56       3596730.6     10441876.22
      3597112.03     10442037.95      3597522.03     10442396.85
#Sta/Elev= 30
  4238.4  420.79  4284.4  417.07  4298.7  417.82  4348.1  415.16  4419.7  413.87
    4512  410.17    4568  406.36  4668.2  397.52  4902.5   392.1  4968.2  392.53
  4978.1  391.09  4986.4  387.92  4991.8   387.7  4993.9  385.45  4994.4  384.95
  5005.7  385.45  5015.5   386.8  5021.6  389.46  5039.2  391.97  5130.2  389.95
  5168.4  391.69  5197.5  390.22    5208  391.09  5297.6  394.01    5364  397.59
  5569.1  411.75  5611.8  415.96  5689.6   420.7    5775  422.04  5870.5  421.74
#Mann= 5 ,-1 , 0
  4238.4      .1       0  4902.5     .16       0  4993.9     .07       0
  5005.7     .16       0    5208     .05       0
Bank Sta=4968.2,5039.2
XS Rating Curve= 0 ,0
Exp/Cntr=0.3,0.1

Type RM Length L Ch R = 1 ,14525   ,831,831,831
BEGIN DESCRIPTION:
UNT0277 IN DUCK CR 9 0
END DESCRIPTION:
XS GIS Cut Line= 4
      3596011.87     10441886.66      3596371.22      10442428.3
      3596496.22     10442605.39      3596807.89     10442823.55
#Sta/Elev= 30
  4253.4  414.19  4266.6  413.22  4351.4  404.75  4408.5  403.41  4435.3  401.22
  4480.7  397.83    4490  396.17  4546.8  392.08  4604.1  391.14  4610.9  391.01
  4805.5  389.25  4892.7  389.74  4919.7  391.08  4964.1  389.51  4970.2  386.48
  4978.9  386.31  4993.9  383.29  4994.4  382.79  5005.7  383.29  5005.9  384.18
  5020.7     388  5035.5  389.99  5052.9  390.66  5100.8  391.21  5157.5  394.79
  5243.9  402.25  5273.5  403.17  5405.4  412.74  5444.7  416.71  5500.6  419.61
#Mann= 11 ,-1 , 0
  4253.4     .05       0  4266.6      .1       0  4435.3     .05       0
    4490      .1       0  4604.1     .16       0  4610.9      .1       0
  4805.5     .16       0  4993.9     .07       0  5005.7     .16       0
  5052.9      .1       0  5405.4     .05       0
Bank Sta=4964.1,5035.5
XS Rating Curve= 0 ,0
Exp/Cntr=0.3,0.1

Type RM Length L Ch R = 1 ,13694   ,238,238,238
BEGIN DESCRIPTION:
UNT0277 IN DUCK CR 8 0
END DESCRIPTION:
XS GIS Cut Line= 4
      3594610.81     10442542.89      3595678.52     10442844.97
      3595944.14     10443006.43      3596448.27     10443099.98
#Sta/Elev= 30
  3795.6  422.48  3838.5  422.62  3890.5  420.42    3932  420.43  3957.2   418.8
  4030.3  411.59  4064.2  405.61  4233.4  390.11  4249.6  387.36    4275  389.81
  4295.8  390.07  4474.1  387.28  4621.3  386.96  4711.5  385.93  4868.5   386.4
  4979.6  387.22    4995  381.33  4995.5  380.83  5006.8  381.33  5014.7  383.75
  5037.7  386.87    5154  388.54  5202.5  391.87  5328.9  397.52  5427.6  398.84
  5492.5  403.91  5508.9  408.31  5529.3  407.63  5580.1   410.9  5728.8  413.98
#Mann= 5 ,-1 , 0
  3795.6     .05       0  4621.3      .1       0  4868.5     .05       0
    4995     .03       0  5006.8     .05       0
Bank Sta=4979.6,5037.7
XS Rating Curve= 0 ,0
Exp/Cntr=0.3,0.1

Type RM Length L Ch R = 1 ,13456   ,149,149,149
BEGIN DESCRIPTION:
UNT0277 IN DUCK CR 6 0
END DESCRIPTION:
XS GIS Cut Line= 3
      3594669.78     10442875.84      3596015.28     10443179.67
      3596427.36     10443253.41
#Sta/Elev= 30
  4005.9   417.8  4054.7  417.83    4099  415.03  4146.2   409.8  4189.4  403.86
  4232.6  400.27  4324.1  394.38  4329.3  395.01  4372.5  390.85  4420.8  389.93
  4469.6  387.07  4500.4  386.29  4550.4  387.44  4807.9  385.63  4879.7  386.57
  4982.2   385.7  4992.5  382.36  4996.8  381.98  4997.3  381.48  5008.6  381.98
  5013.2  385.84  5074.5  385.75  5105.2  387.68    5186  390.19  5269.2     394
  5426.3  403.45  5480.1  407.91  5592.7  406.43  5717.3   411.3  5803.9  412.49
#Mann= 4 ,-1 , 0
  4005.9     .05       0    4099     .08       0  4996.8     .07       0
  5008.6     .08       0
Bank Sta=4982.2,5013.2
XS Rating Curve= 0 ,0
Exp/Cntr=0.3,0.1

Type RM Length L Ch R = 1 ,13307   ,298,298,298
BEGIN DESCRIPTION:
UNT0277 IN DUCK CR 32 0
END DESCRIPTION:
XS GIS Cut Line= 4
      3594661.07     10443125.42      3595010.51      10443097.2
      3595815.63     10443283.83        3596126.     10443466.15
#Sta/Elev= 30
  4061.8  413.98  4143.1  413.32  4303.6  402.42  4363.8  399.55  4385.4  397.75
  4452.1  391.57  4485.9  387.53  4526.9  385.69  4557.7  386.41  4639.8  385.21
  4752.8  384.67  4936.9  387.01  4968.3  386.05  4989.8  383.87  4993.2  380.71
  4993.7  380.21  5004.5  380.21    5005  380.71  5009.4  384.67  5019.7  386.13
  5101.8  386.93  5183.9  389.95  5208.3  391.62  5263.7  397.11  5301.1  400.02
    5387   408.3  5408.7  409.47    5467  414.53  5525.6  416.54  5598.8  415.86
#Mann= 5 ,-1 , 0
  4061.8     .05       0  4385.4     .08       0  4993.2     .07       0
    5005     .08       0  5263.7     .05       0
Bank Sta=4968.3,5019.7
XS Rating Curve= 0 ,0
Exp/Cntr=0.3,0.1

Type RM Length L Ch R = 1 ,13009   ,788,788,788
BEGIN DESCRIPTION:
UNT0277 IN DUCK CR 21 0
END DESCRIPTION:
XS GIS Cut Line= 4
      3594725.39     10443313.72      3595407.68     10443412.68
      3595574.35     10443563.72      3595892.07     10443591.64
#Sta/Elev= 30
  4195.6  412.94  4252.9  412.49    4287  410.38  4323.6  407.34  4352.1  404.22
  4357.2  404.23  4422.3  397.14  4492.5  390.39  4576.3  385.79  4677.3  384.26
  4697.5  384.42  4703.1  385.03  4798.6  384.79  4922.7  386.27  4979.5  385.66
  4993.7  381.37  4994.5  379.31    4995  378.81  5005.8  378.81  5006.3  379.31
  5014.6  383.05  5028.8  385.01    5043  385.92    5110   386.3  5167.9  389.38
  5260.4  397.55  5367.8  408.17  5372.8  408.06  5408.9  412.55  5428.9  413.57
#Mann= 3 ,-1 , 0
  4195.6     .05       0  4994.5     .03       0  5006.3     .05       0
Bank Sta=4979.5,5028.8
XS Rating Curve= 0 ,0
Exp/Cntr=0.3,0.1

Type RM Length L Ch R = 1 ,12221   ,419,419,419
BEGIN DESCRIPTION:
UNT0277 IN DUCK CR 22 0
END DESCRIPTION:
XS GIS Cut Line= 3
      3594534.21      10443814.3      3595448.27      10444186.7
      3596112.31     10443863.79
#Sta/Elev= 30
  4510.2  409.59  4651.3  401.17  4699.4  396.79  4783.3     393  4822.6  390.03
  4896.7  383.51  4942.9  382.42  4966.9  383.93    4983  382.67  4990.4  378.88
  4990.9  378.38  5002.4  378.88    5015  382.77  5026.2  384.33  5234.4  382.68
    5455  384.32  5541.7  387.25  5590.7  386.97  5609.4  386.29  5729.6  390.88
  5795.4  393.53  5868.6  401.38  5908.1  403.79  5913.7  405.28  6043.5  412.25
    6049  413.96  6058.7  413.47  6094.1  414.78  6154.5  414.47  6235.6  414.46
#Mann= 10 ,-1 , 0
  4510.2     .05       0  4783.3      .1       0  4822.6     .05       0
  4990.4     .03       0  5002.4     .05       0    5455     .16       0
  5590.7     .05       0  5729.6     .16       0  6058.7     .05       0
  6154.5     .16       0
Bank Sta=4983,5015
XS Rating Curve= 0 ,0
Exp/Cntr=0.3,0.1

Type RM Length L Ch R = 1 ,11802   ,242,242,242
BEGIN DESCRIPTION:
UNT0277 IN DUCK CR 1 0
END DESCRIPTION:
XS GIS Cut Line= 3
       3594409.2     10444030.45      3595349.31      10444814.3
      3596187.53     10444949.67
#Sta/Elev= 30
  4469.6  411.54  4600.6  409.88  4834.9  388.73  4870.1  387.78  4933.9  382.43
  4976.8  382.73  4997.6  379.17  5019.8  382.95  5075.7  381.87  5153.8  383.08
  5168.2  381.73  5176.5  378.92  5188.5  378.92  5196.8  381.47  5239.7  383.62
  5388.1  381.67  5459.7  383.22  5510.6  386.27  5521.5  386.75  5651.1   395.5
  5747.1  404.73  5797.8  405.71  5878.8  402.32  5980.1  406.79  6096.3  408.82
  6270.8  403.91  6324.5  403.78  6352.1  405.82    6446  413.33  6542.7  416.03
#Mann= 7 ,-1 , 0
  4469.6     .05       0  4976.8     .03       0  5019.8     .16       0
  5510.6      .1       0  5521.5     .16       0  6096.3      .1       0
  6352.1     .16       0
Bank Sta=4976.8,5019.8
XS Rating Curve= 0 ,0
Exp/Cntr=0.3,0.1

Type RM Length L Ch R = 1 ,11560   ,587,587,587
BEGIN DESCRIPTION:
BUCK CREEK 4 0
END DESCRIPTION:
XS GIS Cut Line= 4
      3594340.31     10444139.15      3594631.99     10444514.17
      3594754.39     10444696.46      3595296.05     10445042.82
#Sta/Elev= 30
  4481.4   411.6  4584.9  410.57    4784  401.02  4819.3  397.95  4833.7  397.59
    4898     392    4945  386.18  4952.5  383.76  4977.5  380.74  4989.6  377.39
  4992.6  377.36  4993.1  376.86  5004.6  377.36  5013.6  380.45  5061.9  381.72
  5157.6  382.69  5256.5  382.09  5271.7  382.71  5329.3  380.75    5387  381.04
  5438.4  382.77  5526.3  389.16  5570.3  393.15  5641.3   401.7  5714.1  404.16
  5781.4  408.82  5799.2  409.27    5808   408.6  5813.7  409.81    5819  409.81
#Mann= 7 ,-1 , 0
  4481.4     .05       0    4945     .16       0  4992.6     .07       0
  5004.6     .16       0  5570.3      .1       0  5781.4     .16       0
  5799.2      .1       0
Bank Sta=4977.5,5013.6
XS Rating Curve= 0 ,0
Exp/Cntr=0.3,0.1

Type RM Length L Ch R = 1 ,10973   ,508,508,508
BEGIN DESCRIPTION:
BUCK CREEK 3 1
END DESCRIPTION:
XS GIS Cut Line= 3
      3594132.58      10444657.6      3594424.25      10445092.5
      3595304.42     10445490.92
#Sta/Elev= 30
  4688.9  403.28  4770.4  396.94  4836.4  387.68  4893.5  381.84  4922.5   380.1
  4980.5  382.02  4986.5   380.7  5001.1   376.1  5001.6   375.6    5014   376.1
  5016.5  378.69  5022.5  380.91  5049.6  381.42  5145.6  381.28  5270.8  379.63
  5385.8  380.17    5438  383.25  5466.6  384.04  5512.8  388.04  5564.5  389.59
  5594.4  391.73  5624.8  392.11  5633.8  392.45  5639.3  391.73  5662.4  392.55
  5808.5   399.1  5875.8  403.38  5950.6  406.67  6077.4  414.84  6178.7   417.6
#Mann= 6 ,-1 , 0
  4688.9     .05       0  5001.1     .03       0    5014     .05       0
  5049.6      .1       0  5624.8     .16       0  5808.5      .1       0
Bank Sta=4986.5,5022.5
XS Rating Curve= 0 ,0
Exp/Cntr=0.3,0.1

Type RM Length L Ch R = 1 ,10465   ,475,475,475
BEGIN DESCRIPTION:
BUCK CREEK 19 0
END DESCRIPTION:
XS GIS Cut Line= 3
      3593674.22     10444764.33      3593960.71     10445204.48
      3594163.54     10446067.81
#Sta/Elev= 30
  4700.3  402.96  4864.1  391.78  4876.3  389.82    4979  380.92  5000.2  375.42
  5000.9  375.21  5001.4  374.71  5013.8  375.21  5015.2  379.14  5021.2  380.61
  5078.9  380.39  5114.8   379.1  5123.9  380.61  5129.9  379.34  5174.4  377.86
  5217.5  379.84  5263.6  378.77  5425.6  378.94  5551.3  386.64  5600.4  388.76
    5654  388.95  5737.8  392.91  5808.1  397.72  5859.4  398.93  5931.3  403.22
    5955  404.06  5992.3  402.42  5997.4  403.54  6013.5  402.87  6112.3  408.34
#Mann= 4 ,-1 , 0
  4700.3     .05       0  5000.2     .16       0  5000.9     .03       0
  5013.8     .16       0
Bank Sta=4979,5021.2
XS Rating Curve= 0 ,0
Exp/Cntr=0.3,0.1

Type RM Length L Ch R = 1 ,9990    ,1163,1163,1163
BEGIN DESCRIPTION:
BUCK CREEK 18 0
END DESCRIPTION:
XS GIS Cut Line= 3
      3593309.68      10445019.6      3593684.67     10445610.73
      3593650.88     10446117.57
#Sta/Elev= 30
  4706.9  401.88  4768.5  397.74  4796.8  394.44    4812   391.3  4854.4  387.09
  4869.6  384.82  4942.5  379.23  4971.2  379.97  4984.9  380.08  4993.5  377.57
  4993.7  375.06  4994.2  374.56  5006.6  375.06  5021.3  379.61  5088.2  377.58
  5172.9  377.42  5188.2  377.59  5203.5  379.63  5218.5  378.69  5258.3  380.01
  5276.3   380.7  5297.5  384.11  5318.7  385.14  5339.8  387.82  5404.5   393.1
  5455.6   396.1  5521.9  398.84  5628.3  406.01  5667.2  407.32  5914.9  411.14
#Mann= 7 ,-1 , 0
  4706.9     .05       0  4971.2     .12       0  4993.7     .07       0
  5006.6     .12       0  5258.3     .16       0  5297.5      .1       0
  5455.6     .16       0
Bank Sta=4984.9,5021.3
XS Rating Curve= 0 ,0
Exp/Cntr=0.3,0.1

Type RM Length L Ch R = 1 ,8827    ,1127,1127,1127
BEGIN DESCRIPTION:
BUCK CREEK 17 0
END DESCRIPTION:
XS GIS Cut Line= 3
      3592406.02     10444725.32      3592467.11     10445766.64
      3592853.92     10446506.52
#Sta/Elev= 30
  4075.2  400.42  4076.1   400.3  4161.7  391.95  4281.9  378.18  4339.1  377.22
  4402.1  376.55  4442.1  377.38  4638.8  375.16  4702.6  374.18  4820.1   374.4
    4923  375.68  4983.1  378.26  4993.1  376.19  4996.6  373.63  4997.1  373.13
  5009.7  373.63  5023.1  377.35  5033.2  377.97  5134.7  375.35  5278.5  374.19
  5302.4  374.21  5458.2  375.53  5518.9  379.48  5675.4  392.12    5801   404.5
  5829.9   408.6  5835.5  408.26    5852  409.98    5874  409.98  5953.2   416.3
#Mann= 10 ,-1 , 0
  4075.2     .05       0  4076.1     .16       0  4339.1     .05       0
  4638.8      .1       0  4820.1     .05       0  4996.6     .03       0
  5009.7     .05       0  5278.5      .1       0  5302.4     .05       0
  5458.2     .16       0
Bank Sta=4983.1,5033.2
XS Rating Curve= 0 ,0
Exp/Cntr=0.3,0.1

Type RM Length L Ch R = 1 ,7700    ,741,741,741
BEGIN DESCRIPTION:
BUCK CREEK 16 0
END DESCRIPTION:
XS GIS Cut Line= 3
      3591559.67     10444806.06      3591564.88     10445540.42
      3591411.42      10446838.3
#Sta/Elev= 30
  4400.4  397.62    4456  396.76    4639  381.85    4726  373.38    4896  373.28
  4933.6  374.31    4996  376.52    5006  375.63    5046  376.33  5186.4  372.91
  5289.1  373.06  5438.1  371.83  5599.2  371.62  5630.6  372.28  5879.2   370.5
  5894.8  369.62  5921.4  370.45  5973.1  370.33  6032.2  370.66  6102.7  372.51
  6150.7  372.35  6183.3   373.9  6203.4  375.97  6220.7  375.49  6243.7  377.13
  6308.6  383.08  6334.3  387.87  6391.5  392.79  6414.9  393.74  6441.7  393.52
#Mann= 7 ,-1 , 0
  4400.4     .16       0    4639     .12       0  4933.6     .16       0
    4996     .07       0    5046     .16       0  5973.1     .12       0
  6150.7     .05       0
Bank Sta=4996,5046
XS Rating Curve= 0 ,0
Exp/Cntr=0.3,0.1

Type RM Length L Ch R = 1 ,6959    ,777,777,777
BEGIN DESCRIPTION:
BUCK CREEK 14 0
END DESCRIPTION:
XS GIS Cut Line= 3
        3590893.     10444790.46      3590867.11     10445616.64
      3590629.98     10446740.92
#Sta/Elev= 30
    4262  409.69  4303.2  406.75  4363.2  396.79  4403.3  392.49  4449.2  386.38
  4454.2  387.14  4503.3   381.7  4543.3  378.95  4567.7  376.38  4613.4  373.09
  4710.3  373.19  4943.5  373.39  4983.5  374.34  5003.5  373.45  5023.6  374.64
  5298.1  369.07  5461.6  368.76  5576.2  369.03  5670.6  373.08  5715.3  376.39
  5809.1  380.85  5864.6  384.73  5901.1  385.82  5914.4  387.01  5952.2  387.83
  5964.2  388.84  6053.5  389.74  6064.6  390.66  6103.3  391.13  6237.6   395.6
#Mann= 5 ,-1 , 0
    4262      .1       0  4567.7     .05       0  4710.3     .16       0
  4983.5     .07       0  5023.6     .05       0
Bank Sta=4983.5,5023.6
XS Rating Curve= 0 ,0
Exp/Cntr=0.3,0.1

Type RM Length L Ch R = 1 ,6182    ,750,750,750
BEGIN DESCRIPTION:
BUCK CREEK 13 0
END DESCRIPTION:
XS GIS Cut Line= 4
       3589965.9      10445230.5       3590205.5     10445678.44
      3590468.52     10445795.62      3590583.05     10446717.09
#Sta/Elev= 30
    4311  396.75  4403.5  391.78  4455.7  387.03  4545.8   378.3  4611.6  374.66
  4627.9  372.91  4671.8  370.79  4694.9  371.51  4705.4  371.67  4775.8  372.54
  4788.6   373.4  4924.8  371.24  4939.3  369.84  4959.2  369.54  5023.3  370.11
  5055.5  369.01  5136.6  368.76  5149.8  368.76  5395.2  368.83  5420.1  370.06
  5425.4  371.12  5500.9  376.84  5581.7  384.78  5626.9  387.96  5662.6  392.86
  5737.8  397.84  5818.4  398.55  5838.5   397.5  5910.2  396.74  6035.5  397.27
#Mann= 7 ,-1 , 0
    4311     .05       0  4455.7     .16       0  4694.9      .1       0
  4705.4     .16       0  4959.2     .05       0  5136.6    .033       0
  5149.8     .05       0
Bank Sta=4924.8,5425.4
XS Rating Curve= 0 ,0
Exp/Cntr=0.3,0.1

Type RM Length L Ch R = 1 ,5432    ,444,444,444
BEGIN DESCRIPTION:
BUCK CREEK 11 0
END DESCRIPTION:
XS GIS Cut Line= 3
      3589742.11     10445341.66      3590001.43     10446141.84
       3590522.3     10446704.38
#Sta/Elev= 30
    4055  398.15  4118.1  396.99  4160.1  394.39  4271.3  380.94  4338.1  373.74
  4370.3  370.82  4394.3  370.23  4593.3  372.61  4667.2  372.02  4707.8  371.69
  4747.9  371.58  4801.3  372.87  4843.4  371.41  4891.1  371.88  4946.1  371.81
  4967.1  371.14  4974.5  370.18  4981.3  368.18  4988.8  367.67  4989.3  367.17
  5002.1  367.67  5009.6  368.26    5017   369.9  5186.5  378.61  5299.9  383.53
  5320.9  385.17  5462.6  390.64  5497.8  392.82  5554.5  394.61  5662.8  396.48
#Mann= 9 ,-1 , 0
    4055     .05       0  4271.3      .1       0  4338.1     .05       0
  4394.3      .1       0  4667.2     .16       0  4707.8      .1       0
  4891.1     .05       0  4988.8     .03       0  5002.1     .05       0
Bank Sta=4974.5,5017
XS Rating Curve= 0 ,0
Exp/Cntr=0.3,0.1

Type RM Length L Ch R = 1 ,4988    ,92,92,92
BEGIN DESCRIPTION:
Mapping XS 2918efaf
END DESCRIPTION:
XS GIS Cut Line= 4
       3589325.5     10445818.23      3589622.34     10446122.88
      3589705.67     10446458.82      3590011.86     10446848.04
#Sta/Elev= 30
  4116.8  383.95  4123.8  383.04  4145.1  382.45  4187.6  379.47  4265.3  372.37
  4300.7  371.22  4314.9  370.05  4321.9  367.55  4329.4  365.73  4342.7  365.73
  4343.2  367.33  4357.3  370.78  4371.5  371.57  4399.8  370.79  4551.2  369.36
  4688.4  369.62  4736.6  368.71  4819.1  369.51  4887.2  369.02  4980.9   369.3
  4987.5  368.59  5016.4  367.83  5037.2  368.63    5058  368.65  5072.4  369.51
    5095  370.85  5165.5     373  5279.3  377.74  5349.9  385.03  5383.5  387.12
#Mann= 3 , 0 , 0
  4116.8     .05       0  4980.9     .03       0  5072.4     .05       0
Bank Sta=4980.9,5072.4
XS Rating Curve= 0 ,0
Exp/Cntr=0.3,0.1

Type RM Length L Ch R = 1 ,4896    ,534,534,534
BEGIN DESCRIPTION:
BUCK CREEK 10 0
END DESCRIPTION:
XS GIS Cut Line= 4
      3589281.17     10445891.08      3589559.84     10446177.57
      3589624.95     10446490.07      3589934.42     10446867.16
#Sta/Elev= 30
  4181.6  386.96  4203.9  385.72  4246.3  381.69  4274.6  378.15  4295.7  374.39
    4324  371.23  4387.8  370.82  4401.9  366.58  4416.1  368.65  4423.1  370.76
  4430.2  370.93  4529.2  369.09  4605.9  369.75  4949.5  368.57  4970.3  366.76
  4992.5  367.05  4999.4  366.05  4999.9  365.55  5012.7  366.05  5013.3  366.91
  5019.8  366.51  5034.2  367.69  5070.7  367.36  5077.2  369.23  5141.1  370.85
  5219.3  374.07  5268.8   377.3  5311.9  381.11  5318.3  380.63  5388.3  384.49
#Mann= 3 ,-1 , 0
  4181.6     .05       0  4999.4     .03       0  5012.7     .05       0
Bank Sta=4949.5,5077.2
XS Rating Curve= 0 ,0
Exp/Cntr=0.3,0.1

Type RM Length L Ch R = 1 ,4362    ,584,584,584
XS GIS Cut Line= 2
     3589242.754    10445875.165     3589392.076    10447393.058
#Sta/Elev= 30
       0   388.5   39.81  387.48   99.53  384.33  129.38  381.65  169.19  377.15
  218.96  370.65  228.91  369.91  268.72  369.84  298.58  370.62  308.53  370.32
  318.48  367.96  328.43  366.51  348.34  370.12  418.01  368.55  487.67  367.85
   796.2  367.19  975.35  365.31   985.3  364.79 1005.21  365.63 1035.06  365.28
 1064.92   366.5 1094.78  368.76 1114.68   370.7 1134.59  371.94 1154.49   374.2
 1263.97  382.59  1383.4  393.91 1403.31   395.4 1453.07  400.56 1482.93  402.68
#Mann= 3 , 0 , 0
       0     .05       0  308.53     .03       0  348.34     .05       0
Bank Sta=308.53,348.34
XS Rating Curve= 0 ,0
Exp/Cntr=0.3,0.1

Type RM Length L Ch R = 1 ,3778    ,697,697,697
BEGIN DESCRIPTION:
BUCK CREEK 9 0
END DESCRIPTION:
XS GIS Cut Line= 3
       3589223.9     10445862.48      3589114.53     10446281.74
      3588604.11     10446922.37
#Sta/Elev= 30
  4193.6  388.22  4213.4  388.09  4265.2  384.06  4306.4  382.94  4335.8  380.91
  4381.5  376.62  4416.8  371.79  4451.1     369  4471.8  368.67  4554.4  370.63
  4573.5  364.44  4578.7  365.46  4585.5  368.45  4595.8   370.5  4607.4  370.27
  4770.5  367.98  4892.2  367.93  4977.1  365.99  4984.8  364.15  4991.3  360.22
  4991.8  359.72  5004.6  360.22  5005.9  362.84  5012.3  365.21  5020.3  365.78
  5098.8  370.57  5332.6  394.65  5382.3  398.79  5390.3  398.51    5446  401.65
#Mann= 4 ,-1 , 0
  4193.6     .05       0  4607.4     .16       0  4991.3     .07       0
  5004.6     .16       0
Bank Sta=4977.1,5020.3
XS Rating Curve= 0 ,0
Exp/Cntr=0.3,0.1

Type RM Length L Ch R = 1 ,3081    ,796,796,796
BEGIN DESCRIPTION:
BUCK CREEK 7 0
END DESCRIPTION:
XS GIS Cut Line= 3
      3588528.62      10445529.1       3588348.9     10445737.46
      3588286.45     10446627.41
#Sta/Elev= 30
  4241.2  385.97  4290.1  382.41  4304.4  383.73  4345.2  381.57    4425  377.31
  4453.6   374.9  4473.3   372.2  4487.9  370.23  4515.8  366.93  4580.7  363.96
  4600.8  365.03    4775  367.36  4851.4  368.21  4871.4  365.83  4901.5  367.45
  4973.6  365.76  4981.7  364.34  4991.7  359.47  4995.1  356.47  4995.6  355.97
  5008.4  356.47  5011.8  358.53  5031.8  366.69  5041.8  368.53  5162.1  379.24
  5202.2  381.33  5232.3  384.53  5256.8   385.4  5342.6  392.02  5408.5  395.09
#Mann= 7 ,-1 , 0
  4241.2      .1       0  4345.2     .16       0  4473.3      .1       0
  4487.9     .05       0    4775     .16       0  4995.1     .07       0
  5008.4     .16       0
Bank Sta=4973.6,5031.8
XS Rating Curve= 0 ,0
Exp/Cntr=0.3,0.1

Type RM Length L Ch R = 1 ,2285    ,730,730,730
BEGIN DESCRIPTION:
BUCK CREEK 6 0
END DESCRIPTION:
XS GIS Cut Line= 2
       3587356.7     10445687.94       3587726.5     10446781.72
#Sta/Elev= 30
  4203.9  383.38  4209.1  383.52  4260.6  379.57  4292.3  375.91  4298.2  374.65
  4323.9  373.01  4329.6  371.27  4355.6  368.47  4361.1  367.27  4408.4  363.14
  4607.4  364.53  4638.8  363.37  4644.1  363.99  4670.2  363.33  4682.8  364.04
  4764.6  364.86  4841.2  363.97  4978.4   363.7    4990  359.98  4999.5   354.9
  5003.9  353.32  5016.2  353.32  5021.4  360.14  5031.2  365.36  5047.6  367.92
  5073.4  369.53    5079  370.45  5210.6  381.81  5262.4  385.34  5358.5  389.03
#Mann= 3 , 0 , 0
  4203.9      .5       0  4978.4     .03       0  5031.2     .05       0
Bank Sta=4978.4,5031.2
XS Rating Curve= 0 ,0
Exp/Cntr=0.3,0.1

Type RM Length L Ch R = 1 ,1555    ,353,353,353
BEGIN DESCRIPTION:
BUCK CREEK 3 0
END DESCRIPTION:
XS GIS Cut Line= 3
      3586807.24     10445930.19      3586885.36     10446549.96
      3587317.09     10446916.63
#Sta/Elev= 30
  4271.7  377.88  4333.6  375.19  4404.2  368.08    4430  364.56  4464.7   361.4
  4484.8  358.59    4505  360.05  4535.2  360.13  4565.5  361.11  4676.3  360.77
  4706.6  360.14  4797.3  361.51  4966.4  361.95  4972.9  360.99  4980.7  358.53
  4987.2  356.03  4995.4  351.75  5007.7  351.75  5008.2  352.25  5009.2  354.79
  5023.3  360.34  5036.6  361.98  5150.9  362.54  5285.7  370.09  5321.1  370.65
  5370.6  372.79  5384.8  372.49    5442  374.28  5448.5  374.93  5462.8  374.64
#Mann= 3 , 0 , 0
  4271.7     .05       0  4966.4     .03       0  5036.6     .05       0
Bank Sta=4966.4,5036.6
XS Rating Curve= 0 ,0
Exp/Cntr=0.3,0.1

Type RM Length L Ch R = 1 ,1202    ,630,630,630
BEGIN DESCRIPTION:
BUCK CREEK 2 0
END DESCRIPTION:
XS GIS Cut Line= 3
     3586736.269    10445995.156      3586682.23     10446940.59
      3587337.84      10446956.2
#Sta/Elev= 30
 3844.51  373.01 3983.86  360.84 4023.67  359.11 4063.49  360.57 4143.12  360.57
 4212.79  359.26 4401.91  360.36 4431.77  359.61 4561.17  361.86 4610.94  359.95
 4670.66  360.32 4690.56  361.29 4770.19  368.62    4810  370.13    4830  369.37
    4950  360.45    4980  357.09    4990  353.95  4993.9  351.32  5006.2  351.32
    5010  353.73    5020  356.82  5039.7  360.19  5130.1  361.59  5200.1  365.19
  5230.1  367.53  5280.1  369.63  5380.1  376.17  5410.2   377.1  5445.9   376.7
#Mann= 3 , 0 , 0
 3844.51     .05       0    4950     .03       0  5039.7     .05       0
Bank Sta=4950,5039.7
XS Rating Curve= 0 ,0
Exp/Cntr=0.3,0.1

Type RM Length L Ch R = 1 ,572     ,0,0,0
BEGIN DESCRIPTION:
BUCK CREEK 1 0
END DESCRIPTION:
XS GIS Cut Line= 5
     3586685.607    10445947.159      3586479.14     10447128.13
      3586794.22      10447573.4      3586967.11     10447566.64
      3587421.11     10447256.18
#Sta/Elev= 30
    3180  372.11 3329.44  360.83 3359.33  359.75 3389.22  359.78 3409.15   358.6
 3468.92  360.65  3608.4  359.15 3747.88  358.84 4016.88  360.84  4146.4  358.73
 4196.21  359.56  4427.7  359.13  4814.7  355.11    4880  355.06    4980  356.46
    4990   353.1  4993.9   349.8  5006.2   349.8    5010  353.06    5020  356.17
  5100.1  354.64  5299.5  355.32  5386.1  359.61  5457.9  364.27  5478.9  366.68
  5544.6  370.69  5550.7   371.7  5601.5  374.12  5616.4  373.64  5655.1   374.8
#Mann= 3 , 0 , 0
    3180     .05       0    4980     .03       0    5020     .05       0
Bank Sta=4980,5020
XS Rating Curve= 0 ,0
Exp/Cntr=0.3,0.1

Chan Stop Cuts=-1
Use User Specified Reach Order=0
Composite Channel Slope=5
