--- CARTERS CREEK.prj (project) ---

Proj Title=CARTERS CREEK Base Level Engineering
Current Plan=p01
Default Exp/Contr=0.3,0.1
English Units
Geom File=g01
Flow File=f01
Plan File=p01
Y Axis Title=Elevation
X Axis Title(PF)=Main Channel Distance
X Axis Title(XS)=Station
BEGIN DESCRIPTION:
CARTERS CREEK
END DESCRIPTION:
DSS Export Rating Curves= 0
DSS Export Rating Curve Sorted= 0
DSS Export Volume Flow Curves= 0
DXF OffsetX= 0
DXF OffsetY= 0
DXF ScaleX= 1
DXF ScaleY= 10

--- CARTERS CREEK.p01 (plan) ---

Plan Title=Multiple Run
Short Identifier=Multiple
Geom File=g01
Flow File=f01
Subcritical Flow
K Sum by GR= 0
Std Step Tol= 0.01
Critical Tol= 0.01
Num of Std Step Trials= 20
Max Error Tol= 0.3
Flow Tol Ratio= 0.001
Split Flow NTrial= 30
Split Flow Tol= 0.02
Split Flow Ratio= 0.02
Log Output Level= 0
Friction Slope Method= 1
Unsteady Friction Slope Method= 2
Unsteady Bridges Friction Slope Method= 1
Parabolic Critical Depth
Global Vel Dist=  1 , 1 , 1
Global Log Level= 0
CheckData=True
Encroach Param= -1, 0, 0, 0
BEGIN DESCRIPTION:
Multiple Run
END DESCRIPTION:

--- CARTERS CREEK.f01 (steady flow) ---

Flow Title=Multiple
Program Version=4.10
Number of Profiles= 7
Profile Names=10-year,25-year,50-year,1pct_min,100-year,1pct_plu,500-year
River Rch & RM=CARTERS CREEK,Reach-1         ,114634
     341     443     523     454     614     830     844
River Rch & RM=CARTERS CREEK,Reach-1         ,112219
     387     507     602     524     708     958     982
River Rch & RM=CARTERS CREEK,Reach-1         ,109488
     596     800     965     852    1153    1559    1649
River Rch & RM=CARTERS CREEK,Reach-1         ,108652
     596     800     965     852    1153    1559    1649
River Rch & RM=CARTERS CREEK,Reach-1         ,106777
    1094    1512    1858    1668    2256    3051    3337
River Rch & RM=CARTERS CREEK,Reach-1         ,98481
    1313    1824    2250    2026    2740    3705    4077
River Rch & RM=CARTERS CREEK,Reach-1         ,93119
    2241    3177    3973    3621    4897    6623    7466
River Rch & RM=CARTERS CREEK,Reach-1         ,91351
    2241    3177    3973    3621    4897    6623    7466
River Rch & RM=CARTERS CREEK,Reach-1         ,90412
    2231    3155    3938    3582    4844    6551    7356
River Rch & RM=CARTERS CREEK,Reach-1         ,86047
    2231    3155    3938    3582    4844    6551    7356
River Rch & RM=CARTERS CREEK,Reach-1         ,81317
    2790    3977    4992    4563    6171    8346    9464
River Rch & RM=CARTERS CREEK,Reach-1         ,79519
    2790    3977    4992    4563    6171    8346    9464
River Rch & RM=CARTERS CREEK,Reach-1         ,71382
    3767    5419    6846    6294    8512   11512   13203
River Rch & RM=CARTERS CREEK,Reach-1         ,69930
    4052    5830    7365    6770    9156   12382   14193
River Rch & RM=CARTERS CREEK,Reach-1         ,65235
    4281    6169    7803    7181    9711   13133   15085
River Rch & RM=CARTERS CREEK,Reach-1         ,63285
    4281    6169    7803    7181    9711   13133   15085
River Rch & RM=CARTERS CREEK,Reach-1         ,57762
    4478    6427    8106    7435   10056   13599   15519
River Rch & RM=CARTERS CREEK,Reach-1         ,56352
    4478    6427    8106    7435   10056   13599   15519
River Rch & RM=CARTERS CREEK,Reach-1         ,47068
    5437    7852    9946    9160   12388   16754   19270
River Rch & RM=CARTERS CREEK,Reach-1         ,45126
    5686    8206   10392    9566   12937   17495   20101
River Rch & RM=CARTERS CREEK,Reach-1         ,41414
    5686    8206   10392    9566   12937   17495   20101
River Rch & RM=CARTERS CREEK,Reach-1         ,32860
    5778    8341   10563    9723   13150   17784   20433
River Rch & RM=CARTERS CREEK,Reach-1         ,30803
    6081    8777   11117   10233   13839   18716   21501
River Rch & RM=CARTERS CREEK,Reach-1         ,26682
    6175    8907   11275   10373   14028   18971   21768
River Rch & RM=CARTERS CREEK,Reach-1         ,15728
    6128    8823   11155   10249   13860   18744   21450
River Rch & RM=CARTERS CREEK,Reach-1         ,8640
    6144    8827   11144   10223   13826   18698   21330
Boundary for River Rch & Prof#=CARTERS CREEK,Reach-1         , 1
Up Type= 0
Dn Type= 3
Dn Slope=0.0005
Boundary for River Rch & Prof#=CARTERS CREEK,Reach-1         , 2
Up Type= 0
Dn Type= 3
Dn Slope=0.0005
Boundary for River Rch & Prof#=CARTERS CREEK,Reach-1         , 3
Up Type= 0
Dn Type= 3
Dn Slope=0.0005
Boundary for River Rch & Prof#=CARTERS CREEK,Reach-1         , 4
Up Type= 0
Dn Type= 3
Dn Slope=0.0005
Boundary for River Rch & Prof#=CARTERS CREEK,Reach-1         , 5
Up Type= 0
Dn Type= 3
Dn Slope=0.0005
Boundary for River Rch & Prof#=CARTERS CREEK,Reach-1         , 6
Up Type= 0
Dn Type= 3
Dn Slope=0.0005
Boundary for River Rch & Prof#=CARTERS CREEK,Reach-1         , 7
Up Type= 0
Dn Type= 3
Dn Slope=0.0005
DSS Import GetInterval= 0
DSS Import GetPeak= 0
DSS Import FillOption= 0

--- CARTERS CREEK.g01 (geometry) ---

Geom Title=Existing Conditions
Program Version=4.10

River Reach=CARTERS CREEK   ,Reach-1
Reach XY= 30
      3547364.18      10246177.5      3550766.22     10243154.85
      3549954.89     10241082.93      3552382.72     10239181.29
      3552761.61     10236916.36      3553701.46     10236909.37
      3553488.44     10234839.58      3557475.36     10231426.07
      3558850.54     10228533.79      3558535.88     10226983.17
      3559300.32      10226785.8      3558687.25     10226119.26
      3560449.69     10224950.15      3560673.91     10221152.39
      3563147.12     10218821.67      3567650.03     10217223.49
        3568803.     10214580.78      3572554.65     10212177.99
      3572231.68     10210157.95      3574790.75     10210928.35
       3578653.1     10207264.06      3584035.05     10205866.68
      3584563.32     10204264.68      3586698.71     10204333.69
      3589262.41     10201302.37      3592341.88     10199511.78
      3591913.65     10198576.99      3593277.48      10196662.6
       3599756.5     10197233.47      3604525.59     10199750.35

Type RM Length L Ch R = 1 ,114634  ,369,369,369
BEGIN DESCRIPTION:
CARTERS CREEK 76.0
END DESCRIPTION:
XS GIS Cut Line= 3
      3547932.06     10246217.36       3547441.6     10245622.73
      3546977.23     10245544.61
#Sta/Elev= 30
  4463.3  341.88  4595.3  339.81  4737.4  339.27  4772.5  339.95  4807.7     339
  4829.9  337.87  4854.6  337.41  4879.4  337.96  4900.2  336.85  4928.9  336.46
  4943.2  335.48  4986.2  334.01  4997.6  333.04  5000.3  332.54  5003.6  333.04
  5028.1  334.43  5056.5   334.7    5106  336.53  5120.4  337.38  5140.6  337.18
  5163.4  337.95  5206.4  338.11  5231.6   338.8  5269.9  338.67  5335.6  339.86
  5385.7  339.88  5446.5  340.92  5497.2  340.67  5548.5   341.9    5705  344.58
#Mann= 6 ,-1 , 0
  4463.3     .05       0  4854.6     .16       0  4997.6     .07       0
  5003.6     .16       0  5140.6     .05       0  5548.5      .1       0
Bank Sta=4928.9,5106
XS Rating Curve= 0 ,0
Exp/Cntr=0.3,0.1

Type RM Length L Ch R = 1 ,114265  ,468,468,468
BEGIN DESCRIPTION:
CARTERS CREEK 75.0
END DESCRIPTION:
XS GIS Cut Line= 3
       3548218.5     10245948.23      3547762.78     10245470.82
      3547292.11     10244891.65
#Sta/Elev= 30
  4439.4  340.49  4526.4  339.47    4590  339.84  4646.6  338.42  4674.9  338.52
  4687.8  339.28  4724.6  340.92  4738.7  340.86  4766.7  338.27  4811.3   336.8
  4849.4  336.36  4915.5  334.18  4964.9  335.04    4973  334.54    4979  334.46
  4986.7  333.03  4997.4  331.59  5000.2  331.09  5003.4  331.59  5007.3  332.39
  5021.5  333.21  5077.7  334.35  5092.2  334.68    5284  336.06  5298.4   335.7
  5376.7   337.6  5419.8  337.36  5504.5  338.36  5753.8  343.81  5845.7  346.35
#Mann= 9 ,-1 , 0
  4439.4     .05       0  4687.8      .1       0  4811.3     .05       0
  4849.4      .1       0    4973     .05       0  4986.7      .1       0
  4997.4     .07       0  5003.4      .1       0  5077.7     .05       0
Bank Sta=4964.9,5092.2
XS Rating Curve= 0 ,0
Exp/Cntr=0.3,0.1

Type RM Length L Ch R = 1 ,113797  ,503,503,503
BEGIN DESCRIPTION:
CARTERS CREEK 74.0
END DESCRIPTION:
XS GIS Cut Line= 4
      3548442.11     10245891.65       3548185.2     10245304.43
       3547959.4     10245088.01       3547492.1     10244741.64
#Sta/Elev= 30
    4168  340.74  4211.7  340.86  4229.2  340.46  4316.9   340.1  4479.5  338.49
  4571.9  338.28  4628.6  337.34  4659.6  336.38  4768.3  335.09  4807.8  334.18
  4905.1  333.48  4926.2  332.41  4975.9   331.3  5032.5  331.79  5071.9  330.92
  5074.7  330.42  5077.9  330.92  5089.1  331.58  5103.2  331.16  5116.4  331.61
  5130.8  331.54  5224.5  334.01  5445.7   337.7  5489.5  339.05  5510.4  339.14
  5539.6  340.34  5575.1  341.21  5639.8  342.19  5660.6     343  5703.4  343.79
#Mann= 5 ,-1 , 0
    4168     .05       0  4316.9      .1       0  4628.6     .05       0
  5071.9     .03       0  5077.9     .05       0
Bank Sta=5032.5,5089.1
XS Rating Curve= 0 ,0
Exp/Cntr=0.3,0.1

Type RM Length L Ch R = 1 ,113294  ,327,327,327
BEGIN DESCRIPTION:
CARTERS CREEK 73.0
END DESCRIPTION:
XS GIS Cut Line= 4
      3548614.79     10245483.01      3548403.56     10244986.31
      3548241.52     10244680.02      3547992.12     10244241.66
#Sta/Elev= 30
  4339.8  337.44  4458.5  337.36  4487.6  337.66  4558.5  336.82  4587.6  337.05
  4623.8  335.42  4874.8  332.06  4891.9   331.3  4897.6  331.52  4957.9  330.13
  4993.3  328.82    4996  328.32  4999.3  328.82  5023.9  329.91    5046  329.06
  5062.3  328.88    5134  330.72  5150.3  330.52  5254.1   331.4  5297.3  332.96
  5372.3  334.09  5399.6  334.96  5488.8  336.53  5511.8  337.41  5517.8     338
  5561.1     339  5598.5  340.67  5626.9   341.3  5707.4  344.28  5730.4  344.71
#Mann= 3 ,-1 , 0
  4339.8     .05       0  4993.3     .03       0  4999.3     .05       0
Bank Sta=4957.9,5023.9
XS Rating Curve= 0 ,0
Exp/Cntr=0.3,0.1

Type RM Length L Ch R = 1 ,112967  ,395,395,395
BEGIN DESCRIPTION:
CARTERS CREEK 72.0
END DESCRIPTION:
XS GIS Cut Line= 3
      3548742.11     10245241.66      3548509.75     10244488.18
      3548383.03     10244233.01
#Sta/Elev= 30
    4385  336.65  4471.9  335.63  4504.6  334.96  4531.5  335.01  4562.9  333.66
  4738.5   331.1  4879.6  329.25  4897.8  329.46  4912.2  329.17  4939.7  329.55
  4950.1  328.91    4971  328.41  4999.4  326.72  5002.2  326.22  5005.4  326.72
  5010.2  327.68  5015.5  328.15  5023.4  329.46  5042.9  330.39  5065.2  329.66
  5086.2  329.53  5107.1  329.99    5128  330.92  5159.3  331.58  5214.3  332.95
  5250.1  333.23  5294.9  334.33  5325.9  334.67  5348.3  335.57  5458.4  337.82
#Mann= 5 ,-1 , 0
    4385     .05       0  4738.5      .1       0  4999.4     .07       0
  5005.4      .1       0  5159.3     .05       0
#XS Ineff= 2 ,-1
 4802.95 4929.43  329.56 5042.39  5161.7  330.45
Permanent Ineff=
       F       F
Bank Sta=4939.7,5023.4
XS Rating Curve= 0 ,0
Exp/Cntr=0.3,0.1

Type RM Length L Ch R = 1 ,112572  ,55,55,55
BEGIN DESCRIPTION:
CARTERS CREEK 71.3
END DESCRIPTION:
XS GIS Cut Line= 3
       3549321.8     10245111.04      3548923.13     10244564.98
      3548601.33     10244083.28
#Sta/Elev= 30
  4362.5  329.03  4461.1  329.71  4490.5  329.66  4519.8  328.87  4540.7  329.47
  4584.6  329.17  4626.4  329.83  4712.1  329.47  4770.3  328.54  4812.5  328.89
  4833.4  328.51  4840.5  327.69  4848.1  328.26  4856.5  326.92  4862.7  327.17
  4869.4  326.43  4898.3  326.74  4939.3  326.25    4942  325.75  4945.3  326.25
    4970  326.57  5136.1  326.92  5178.2  326.39  5186.9  327.88  5193.2  329.83
  5199.2  330.25  5244.3  331.83  5322.4  333.57  5430.5  336.86  5617.9  340.42
#Mann= 5 ,-1 , 0
  4362.5     .05       0  4840.5      .1       0  4939.3    .033       0
  4945.3      .1       0    4970     .05       0
#XS Ineff= 2 ,-1
 4345.45 4541.82  329.52 4703.64 4812.73  328.98
Permanent Ineff=
       F       F
Bank Sta=4848.1,5186.9
XS Rating Curve= 0 ,0
Exp/Cntr=0.3,0.1

Type RM Length L Ch R = 1 ,112517  ,57,57,57
BEGIN DESCRIPTION:
CARTERS CREEK 71.2
END DESCRIPTION:
XS GIS Cut Line= 3
      3549408.38     10245158.52      3549009.69     10244612.45
      3548687.85     10244130.69
#Sta/Elev= 30
  4308.5   327.1  4354.2  329.07  4390.3  328.55  4517.7   329.2  4576.4  328.25
  4676.1  329.32  4854.5  327.75  4859.8  326.54  4866.2  324.61  4868.9  324.11
  4872.2  324.61  4875.3  324.71    4890   328.7  4969.6  330.03  5041.5  329.98
  5062.5     329  5069.8  329.58  5092.6  329.32  5113.6  328.77  5119.6  327.45
  5134.6  326.79  5170.7   326.8    5178  327.01  5185.7  328.29  5191.7  327.73
  5200.7  329.19  5206.7   328.8  5257.7  331.27  5380.9  335.11    5564  339.31
#Mann= 5 ,-1 , 0
  4308.5     .05       0  4859.8      .1       0  4866.2     .07       0
  4872.2      .1       0  5062.5     .05       0
#XS Ineff= 2 ,-1
 4301.82 4670.11  329.53    5005 5306.48  330.11
Permanent Ineff=
       F       F
Bank Sta=4854.5,4890
XS Rating Curve= 0 ,0
Exp/Cntr=0.3,0.1

Type RM Length L Ch R = 1 ,112460  ,109,109,109
BEGIN DESCRIPTION:
CARTERS CREEK 71.1
END DESCRIPTION:
XS GIS Cut Line= 3
      3549431.82     10245106.44      3549033.13     10244560.36
      3548711.29     10244078.61
#Sta/Elev= 30
  4365.6  327.47    4405  327.06  4433.5   328.4  4469.9  328.13  4505.4  329.07
  4591.1  327.77  4747.9  328.42  4880.1  326.98  4904.7  326.92  4919.4  325.94
  4941.1  325.51  4945.7  324.59  4948.5  324.09  4951.7  324.59  4954.9  325.51
  4963.4  324.68  4969.6  325.25  4978.1  324.86  4984.3  325.82  4998.9  324.62
  5005.1  325.87  5013.6  325.96  5019.8  326.99  5031.6  325.97  5055.4  326.86
  5064.2   326.5  5076.4  327.39  5208.6  329.23  5445.8  336.35  5621.1   340.1
#Mann= 5 ,-1 , 0
  4365.6     .05       0  4880.1      .1       0  4945.7     .07       0
  4951.7      .1       0  5031.6     .05       0
#XS Ineff= 1 ,-1
 4353.64 4747.27  328.44
Permanent Ineff=
       F
Bank Sta=4919.4,4984.3
XS Rating Curve= 0 ,0
Exp/Cntr=0.3,0.1

Type RM Length L Ch R = 1 ,112351  ,132,132,132
BEGIN DESCRIPTION:
CARTERS CREEK 71.0
END DESCRIPTION:
XS GIS Cut Line= 3
      3549556.62     10245121.87      3549157.95      10244575.8
      3548837.49     10244096.11
#Sta/Elev= 30
  4320.2  331.37  4352.4  330.36  4387.9  330.23  4544.7  327.57  4630.4  328.27
  4789.5  326.68  4875.2  326.35  4896.1  326.78  4939.6  325.66  4981.8  324.24
  4986.1  322.32  4988.8  321.82  4992.1  322.32  4995.8  324.06  5002.6  322.97
  5011.6  324.27  5017.6  322.49  5032.6   324.5  5038.6  323.85  5047.6  324.73
  5053.6  324.58  5061.4  325.89  5068.6  326.83  5140.7  328.27  5161.8  328.08
  5299.9  330.22  5350.1  332.75  5422.2  333.85  5501.1  336.98  5573.2  338.07
#Mann= 3 ,-1 , 0
  4320.2     .05       0  4986.1     .04       0  4992.1     .05       0
#XS Ineff= 1 ,-1
 4432.27 4629.55  328.54
Permanent Ineff=
       F
Bank Sta=4939.6,5061.4
XS Rating Curve= 0 ,0
Exp/Cntr=0.3,0.1

Type RM Length L Ch R = 1 ,112219  ,361,361,361
BEGIN DESCRIPTION:
CARTERS CREEK 71.4
END DESCRIPTION:
XS GIS Cut Line= 3
      3549643.53     10245038.31      3549244.87     10244492.26
      3548923.06     10244010.56
#Sta/Elev= 30
  4369.5  330.83  4568.3  326.76  4704.2  328.68  4733.6  326.31  4804.6  328.53
  4854.8  326.04  4890.4  327.91    4905  325.81  4940.6  328.98  4961.4  326.92
  4969.9  323.85  4989.1  322.56  5002.4  321.29  5005.2  320.79  5008.4  321.29
  5013.5  322.03    5041  326.19    5062  328.87    5077  327.14  5170.1  329.98
  5286.9  328.59    5359   332.4  5401.4  332.42  5407.4  330.39  5488.4  334.35
  5566.5  334.06  5581.6  336.51  5602.6  334.66  5617.6  337.26  5624.9  335.72
#Mann= 5 ,-1 , 0
  4369.5      .1       0  4989.1     .08       0  5002.4     .07       0
  5008.4     .08       0  5013.5      .1       0
#XS Ineff= 1 ,-1
 4418.18    4940  329.01
Permanent Ineff=
       F
Bank Sta=4961.4,5041
XS Rating Curve= 0 ,0
Exp/Cntr=0.3,0.1

Type RM Length L Ch R = 1 ,111858  ,433,433,433
BEGIN DESCRIPTION:
CARTERS CREEK 70.0
END DESCRIPTION:
XS GIS Cut Line= 3
      3549891.61     10244760.95      3549498.46     10244281.58
      3549291.61     10244060.94
#Sta/Elev= 30
  4503.5  328.75  4559.4  327.95  4616.8  326.26  4651.9  325.91  4687.1  326.18
    4695  325.72  4730.2  325.27  4758.9  325.97  4779.7  325.01  4857.9  324.08
  4872.2  323.49  4900.5  323.96  4929.4  323.96  4956.9  324.56  4979.2  323.39
  4985.6  322.61    4997  319.65  4999.7  319.15    5003  319.65    5007  320.91
  5014.3  322.38  5020.8  322.85  5071.7  322.05  5145.9  323.75  5191.8  325.72
  5266.4   327.2  5354.5   328.8  5368.6   329.8  5382.8  330.17  5425.9  330.46
#Mann= 6 ,-1 , 0
  4503.5     .05       0  4900.5     .12       0    4997     .07       0
    5003     .12       0  5145.9      .1       0  5266.4     .05       0
Bank Sta=4979.2,5020.8
XS Rating Curve= 0 ,0
Exp/Cntr=0.3,0.1

Type RM Length L Ch R = 1 ,111425  ,326,326,326
BEGIN DESCRIPTION:
CARTERS CREEK 69.0
END DESCRIPTION:
XS GIS Cut Line= 3
      3550242.11     10244441.65      3549942.11     10244157.05
      3549642.08     10243891.62
#Sta/Elev= 30
  4584.6   328.5  4598.6  327.66  4634.2  326.66  4648.3  326.72    4688  325.24
  4699.7  325.11    4726  324.45  4740.1  324.74  4761.6  323.52  4789.9  323.89
    4804  323.03  4827.8  322.64  4860.3  322.32  4881.7  321.47  4895.9   321.7
  4931.1  320.98  4980.8  321.15  4987.7  320.43  4994.7  317.55  4998.1  317.55
  4998.8  316.25  5001.5  315.75  5004.8  316.25    5016   321.5  5044.4  320.63
  5065.3  321.53    5108  320.97    5131  321.26    5200     323  5398.7  326.35
#Mann= 7 ,-1 , 0
  4584.6     .05       0    4688     .16       0  4699.7     .05       0
  4827.8     .16       0  4998.8     .07       0  5004.8     .16       0
    5131      .1       0
Bank Sta=4980.8,5016
XS Rating Curve= 0 ,0
Exp/Cntr=0.3,0.1

Type RM Length L Ch R = 1 ,111099  ,334,334,334
BEGIN DESCRIPTION:
CARTERS CREEK 68.0
END DESCRIPTION:
XS GIS Cut Line= 4
       3550442.1     10244141.64      3550202.89     10243953.46
      3549985.87     10243823.25      3549742.11     10243741.64
#Sta/Elev= 30
  4603.9   326.5    4629  325.74  4660.8  325.22  4681.6  323.69  4696.1   324.9
    4725  323.21  4824.4  320.18  4888.5  318.93  4924.1  319.31    4961  318.48
  4982.4  318.59  4994.9   315.3  4997.7   314.8  5000.9   315.3  5003.8  315.65
  5013.5  318.36  5025.8  319.65  5034.9   320.5  5040.7  319.73  5056.3  320.78
  5062.1  319.94  5077.6  319.45  5120.4  320.09  5160.6  321.49  5192.9  321.73
  5276.3  323.79  5302.4  323.58    5334  325.56  5355.1  325.16  5418.4   326.7
#Mann= 5 ,-1 , 0
  4603.9     .05       0    4629     .16       0  4994.9     .07       0
  5000.9     .16       0  5192.9      .1       0
Bank Sta=4982.4,5025.8
XS Rating Curve= 0 ,0
Exp/Cntr=0.3,0.1

Type RM Length L Ch R = 1 ,110765  ,477,477,477
BEGIN DESCRIPTION:
CARTERS CREEK 67.0
END DESCRIPTION:
XS GIS Cut Line= 4
      3550692.11     10244041.65      3550431.65     10243718.86
      3550218.08     10243587.14      3549881.68     10243447.81
#Sta/Elev= 30
  4408.8  330.24  4410.6  330.24  4465.6     329  4473.1  328.38    4480  326.95
  4494.4  326.35  4588.8  324.61  4671.9  323.09  4700.7  323.15  4765.5  319.89
  4843.7  317.44    4865  317.73  4893.5  316.93  4938.4   317.8    4975   316.6
  4980.9  316.09  4987.5   313.9  4999.2  312.39  5001.9  311.89  5005.2  312.39
    5011  315.86  5017.6  316.97  5023.5     316  5046.3  316.01  5081.1  318.52
  5152.7  319.46  5176.6  319.19  5199.7  320.04  5266.3  321.63  5438.6  325.18
#Mann= 8 ,-1 , 0
  4408.8     .05       0  4410.6     .16       0  4588.8      .1       0
  4765.5     .12       0  4999.2     .07       0  5005.2     .12       0
  5199.7     .16       0  5266.3      .1       0
Bank Sta=4975,5017.6
XS Rating Curve= 0 ,0
Exp/Cntr=0.3,0.1

Type RM Length L Ch R = 1 ,110288  ,800,800,800
BEGIN DESCRIPTION:
CARTERS CREEK 66.0
END DESCRIPTION:
XS GIS Cut Line= 4
      3551246.74     10243821.53      3550604.21     10243426.72
      3550383.01      10243226.9      3549992.12     10243241.64
#Sta/Elev= 30
  4075.2  323.16  4369.6  323.74  4433.5  321.97  4618.7  319.95  4638.3  320.12
  4660.2  319.32  4717.6  318.17  4769.7  317.96  4775.6  317.25  4784.9  317.03
  4804.3  317.39  4834.2  316.44  4848.4  316.89    4891  315.99    4962  315.77
  4982.9  315.23  4990.3  313.82  4997.1  313.93  5008.3  312.76    5011  312.26
  5014.3  312.76  5018.7  314.42  5039.7   314.6  5047.1  315.41    5089  317.31
  5096.5  317.73  5117.4  316.87  5155.7  316.94  5208.4  318.62  5518.6  324.05
#Mann= 7 ,-1 , 0
  4075.2     .16       0  4618.7      .1       0  4660.2     .16       0
  4804.3     .12       0  5008.3     .07       0  5014.3     .12       0
  5155.7      .1       0
Bank Sta=4962,5089
XS Rating Curve= 0 ,0
Exp/Cntr=0.3,0.1

Type RM Length L Ch R = 1 ,109488  ,836,836,836
BEGIN DESCRIPTION:
CARTERS CREEK 65.0
END DESCRIPTION:
XS GIS Cut Line= 4
       3551776.2     10242897.03      3551176.61     10242811.04
      3550599.95     10242920.53      3550036.49     10243092.13
#Sta/Elev= 30
  3940.2  328.62  3999.6  328.34  4075.7  328.51    4106   329.5  4217.1  329.45
  4257.5  327.29  4469.7  320.94  4489.9  320.02  4505.7  318.15  4515.1  318.25
  4737.8  317.06  4764.3  319.94  4784.6  319.62    4805  314.87  4822.3  311.15
  4825.1  310.65  4828.3  311.15  4847.4  313.33    4866   313.6  4895.7  313.22
    4978  314.04  4998.4  311.48  5069.6  314.26    5122  314.33  5130.2  314.45
  5226.2  315.17  5330.6  317.56  5466.6  318.68  5538.3  320.61  5721.9  321.99
#Mann= 10 ,-1 , 0
  3940.2     .08       0  3999.6      .1       0  4515.1     .05       0
  4822.3     .07       0  4828.3     .05       0  4895.7     .12       0
    5122     .16       0  5130.2     .12       0  5226.2     .16       0
  5330.6      .1       0
Bank Sta=4805,4866
XS Rating Curve= 0 ,0
Exp/Cntr=0.3,0.1

Type RM Length L Ch R = 1 ,108652  ,1875,1875,1875
BEGIN DESCRIPTION:
CARTERS CREEK 64.0
END DESCRIPTION:
XS GIS Cut Line= 4
      3551642.14     10242541.66        3551212.     10242232.97
      3550453.92     10242241.93      3549506.06     10242871.75
#Sta/Elev= 30
  4081.4  330.26  4148.7  328.45  4272.4  324.71  4630.7  314.69  4710.7  313.49
  4820.7  313.79  4860.8  311.04  4930.8  311.03  4960.8  312.71  4970.8  312.29
  4990.8  310.99  5020.8  311.32  5087.8  310.91  5090.5  310.41  5093.8  310.91
  5140.8  311.96  5290.1  312.75  5831.3  317.67  5839.4  318.43  5918.5  317.63
  5939.5  318.66  5954.6  317.51  5960.6   318.4  5983.5  317.96  5996.7  318.99
  6047.8  318.47  6098.9  320.64  6213.1  319.95    6463  323.65    6507  324.09
#Mann= 9 ,-1 , 0
  4081.4      .1       0  4148.7     .08       0  4272.4     .05       0
  4960.8     .12       0  5020.8     .05       0  5087.8     .04       0
  5093.8     .05       0  5290.1     .08       0    6463     .05       0
Bank Sta=4970.8,5140.8
XS Rating Curve= 0 ,0
Exp/Cntr=0.3,0.1

Type RM Length L Ch R = 1 ,106777  ,659,659,659
BEGIN DESCRIPTION:
CARTERS CREEK 63.0
END DESCRIPTION:
XS GIS Cut Line= 3
       3551792.1     10242341.64      3550138.43     10240729.44
      3549466.56     10240181.94
#Sta/Elev= 30
  2786.6  331.37  2897.7  328.88  3210.9  319.26  3380.6  315.55  3635.2  311.03
  3642.2  311.06  3663.5  314.24  3684.7  311.61    3713  311.08  3748.4  308.88
    4017   308.8  4137.3  312.27    4215  312.69    4314   311.2  4406.1  312.21
  4455.5  311.09  4582.8  311.54  4674.7  309.22  4710.1  310.42  4816.1  309.06
  4950.6  310.26  4985.9  306.54  4999.8   304.9  5028.3  309.07  5035.3  310.39
  5070.7  314.41  5142.3  316.46  5297.8  323.65    5497  328.03  5962.8  332.86
#Mann= 4 ,-1 , 0
  2786.6      .1       0  2897.7     .07       0  4985.9     .05       0
  5035.3     .07       0
#XS Ineff= 1 ,-1
 3484.38 4218.18   312.7
Permanent Ineff=
       F
Bank Sta=4950.6,5028.3
XS Rating Curve= 0 ,0
Exp/Cntr=0.3,0.1

Type RM Length L Ch R = 1 ,106118  ,594,594,594
BEGIN DESCRIPTION:
CARTERS CREEK 61.0
END DESCRIPTION:
XS GIS Cut Line= 4
      3551832.63     10241777.21      3550810.34     10240557.92
      3550647.77     10240310.23      3550313.57      10240123.6
#Sta/Elev= 30
  3224.6  319.88  3449.1  314.74  3619.6   312.4  3648.2  312.59  3917.5  307.61
  4002.1  307.21    4045  306.31  4151.7  307.05  4223.2  306.01  4301.3  306.87
  4322.1  306.82  4342.9  305.84  4379.3  305.89  4406.7  307.11  4492.5  307.33
  4549.8   309.4  4669.5  309.57  4755.3  308.18  4790.5  306.73  4933.9  306.45
    4955  304.51  4991.2  303.27  4997.3  301.96    5000  301.46  5003.3  301.96
  5027.3  305.56  5050.5  306.43  5165.2  307.37  5424.5  320.79  5494.8  323.04
#Mann= 3 ,-1 , 0
  3224.6     .05       0  4997.3     .03       0  5003.3     .05       0
#XS Ineff= 1 ,-1
    3750 4670.45  309.51
Permanent Ineff=
       F
Bank Sta=4933.9,5050.5
XS Rating Curve= 0 ,0
Exp/Cntr=0.3,0.1

Type RM Length L Ch R = 1 ,105524  ,398,398,398
BEGIN DESCRIPTION:
CARTERS CREEK 60.0
END DESCRIPTION:
XS GIS Cut Line= 4
       3552431.6     10241065.42      3551498.46     10240375.33
      3551033.19      10239887.6      3550792.13     10239691.66
#Sta/Elev= 30
  3378.5  320.29  3474.3  319.88  3524.4  318.26  3657.1  315.47  3716.4  314.61
  3745.6  313.08  3831.2  310.73  3902.6  310.16  3957.5  310.07  4024.6  309.44
  4124.1  305.46  4211.2   305.1  4288.3  303.02  4317.6  304.42    4424  304.32
  4474.1  305.27  4532.6  304.76  4581.6  305.28  4645.2     307  4765.3  306.93
  4942.4  303.46  4963.4  303.71  4984.8  301.51  4988.8  300.25  4991.5  299.75
  4994.8  300.25  5041.5  304.15  5154.4  305.03  5374.4  312.79  5523.8  316.81
#Mann= 6 ,-1 , 0
  3378.5     .16       0  3657.1     .05       0  3902.6     .16       0
  3957.5     .05       0  4988.8     .03       0  4994.8     .05       0
Bank Sta=4963.4,5041.5
XS Rating Curve= 0 ,0
Exp/Cntr=0.3,0.1

Type RM Length L Ch R = 1 ,105126  ,557,557,557
BEGIN DESCRIPTION:
CARTERS CREEK 59.0
END DESCRIPTION:
XS GIS Cut Line= 3
      3552531.48     10240935.27      3551414.33     10239711.54
      3550777.93     10239572.37
#Sta/Elev= 30
  3467.4  322.56  3773.7  315.51  4007.5  308.99  4149.3  307.08  4219.6  304.96
  4227.1  305.68  4361.5  305.44  4382.5  304.65  4404.1  305.49  4510.1  304.96
  4552.7  304.41  4587.8  300.68  4595.3  300.75  4609.4  303.31  4644.6   304.5
  4948.6  305.56  4962.8  304.49  4970.2  301.35    4977  300.85  4984.4  298.54
  4995.6   298.5  4998.3     298  5001.6   298.5  5012.8  299.05  5033.7  302.83
  5047.9  303.96  5069.5  305.93  5237.5  306.19    5577  315.34  5775.8  317.72
#Mann= 3 ,-1 , 0
  3467.4     .05       0  4995.6     .04       0  5001.6     .05       0
Bank Sta=4962.8,5047.9
XS Rating Curve= 0 ,0
Exp/Cntr=0.3,0.1

Type RM Length L Ch R = 1 ,104569  ,1605,1605,1605
BEGIN DESCRIPTION:
CARTERS CREEK 58.0
END DESCRIPTION:
XS GIS Cut Line= 5
      3553108.72     10240054.16       3552353.5     10239958.67
      3551857.27     10239411.25      3551242.38     10239368.39
      3550986.75     10239182.08
#Sta/Elev= 30
  3692.7  323.78  4227.3  310.91    4315  309.89  4404.9  306.43  4629.7  307.26
  4721.1  305.56  4835.1  303.68  4856.1  300.53  4962.8  300.88  4990.6  299.46
    4995  297.82  4997.8  297.32    5001  297.82  5054.8  302.98  5183.1  301.87
  5308.2  301.72  5328.3  302.91  5348.3  306.74  5388.4  301.83  5521.8  303.35
  5588.9  305.16    5609  308.21  5659.1  306.41  5729.3  306.86  5799.4  308.76
  5806.8  310.33  5817.6  309.13  5893.5  310.93  5954.8  310.29  6125.5  312.19
#Mann= 9 ,-1 , 0
  3692.7     .05       0  4227.3      .1       0  4721.1     .12       0
    4995     .07       0    5001     .12       0  5183.1     .16       0
  5521.8     .05       0  5817.6     .08       0  5954.8     .05       0
Bank Sta=4962.8,5054.8
XS Rating Curve= 0 ,0
Exp/Cntr=0.3,0.1

Type RM Length L Ch R = 1 ,102964  ,686,686,686
BEGIN DESCRIPTION:
CARTERS CREEK 57.0
END DESCRIPTION:
XS GIS Cut Line= 4
      3552992.12     10239441.66      3552535.79     10238903.98
      3551871.72      10238647.9        3551199.     10238513.36
#Sta/Elev= 30
  4014.4  317.73  4319.2  309.06  4390.6  307.89  4425.8  306.14  4468.6  306.05
  4659.7   301.8    4819  299.52  4916.8  299.16  4970.1  299.38  4980.8  298.19
  4988.2  295.92  4999.2  294.98    5002  294.48  5005.2  294.98  5012.8  297.07
  5023.7  298.51  5034.4  298.78  5218.3  298.25    5313   298.6    5351   299.9
    5442  298.12  5506.6  299.18  5532.9  298.07  5553.3  299.83  5583.9  300.62
  5640.9  300.33    5646  301.15  5737.4  302.84  5837.3  304.28  6117.4  311.07
#Mann= 8 ,-1 , 0
  4014.4     .05       0  4916.8     .12       0  4999.2     .07       0
  5005.2     .12       0  5218.3     .05       0  5506.6     .12       0
  5737.4      .1       0  5837.3     .05       0
Bank Sta=4970.1,5034.4
XS Rating Curve= 0 ,0
Exp/Cntr=0.3,0.1

Type RM Length L Ch R = 1 ,102278  ,627,627,627
BEGIN DESCRIPTION:
CARTERS CREEK 56.0
END DESCRIPTION:
XS GIS Cut Line= 4
      3553342.14     10238841.67      3552535.79     10238257.28
      3551974.81     10238231.19      3551342.08     10238191.64
#Sta/Elev= 30
  3573.9  321.29  3702.7  318.36  3989.6  309.95  4226.2  304.14  4368.4  301.39
    4469   300.4    4528  298.78  4593.5  298.66  4632.2  297.26  4663.5  296.23
  4683.6  294.52  4723.6  296.78  4753.6  297.53  4798.7  297.22  4823.7  297.86
  4883.8  298.07  4943.8  297.87  4953.8  297.13  4973.9  297.36  4983.9  296.52
  4993.9  294.18  5000.9  291.64  5003.6  291.14  5006.9  291.64  5023.9  296.99
  5180.6  298.86  5314.4   302.1  5514.8  305.44  5745.2     312  5765.3  312.16
#Mann= 6 ,-1 , 0
  3573.9     .05       0    4528      .1       0  4632.2     .12       0
  5000.9     .07       0  5006.9     .12       0  5180.6     .05       0
Bank Sta=4973.9,5023.9
XS Rating Curve= 0 ,0
Exp/Cntr=0.3,0.1

Type RM Length L Ch R = 1 ,101651  ,994,994,994
BEGIN DESCRIPTION:
CARTERS CREEK 55.0
END DESCRIPTION:
XS GIS Cut Line= 3
       3553256.3     10238370.15      3552485.38     10237810.33
      3551916.08     10237433.25
#Sta/Elev= 30
  3888.6  314.14  3954.8  312.27  4041.8  310.51  4095.2  308.02  4240.5  302.98
  4360.2  300.25  4485.5  298.16  4562.8  297.53  4589.3  298.03  4627.7  297.31
  4706.1  297.79  4763.8  298.06  4778.5  299.07  4784.7  298.12  4844.7  296.93
  4893.2  294.92  4965.2  295.86    4979  294.59  4988.1   292.4  4991.1  290.19
  4993.8  289.69  4997.1  290.19  5001.2  290.31  5009.1  294.08  5015.1  295.17
  5030.2  295.81  5081.3  295.96  5121.2  297.03  5355.1  303.94  5524.2   306.6
#Mann= 9 ,-1 , 0
  3888.6     .05       0  3954.8      .1       0  4095.2     .05       0
  4360.2      .1       0  4589.3     .16       0  4706.1     .12       0
  4991.1     .07       0  4997.1     .12       0  5121.2     .05       0
Bank Sta=4965.2,5030.2
XS Rating Curve= 0 ,0
Exp/Cntr=0.3,0.1

Type RM Length L Ch R = 1 ,100657  ,807,807,807
BEGIN DESCRIPTION:
CARTERS CREEK 53.0
END DESCRIPTION:
XS GIS Cut Line= 3
       3553492.1     10238091.64      3552887.35     10237467.35
      3551625.76     10236968.78
#Sta/Elev= 30
  3767.8  308.68  4150.9  301.33  4460.9  297.24    4482     298  4667.8  295.69
  4719.7  296.08  4830.1  294.54  4878.8  295.46  4962.6  294.92  4975.9  294.47
  4986.7  292.02  4989.3  288.46  4992.1  287.96  4995.3  288.46  5016.7  293.68
  5046.4  295.08  5086.3  295.06    5363  302.81  5560.6  304.73  5599.6  305.37
  5622.4   303.6  5669.5  303.18  5825.4  303.23  5838.8  304.67  5863.2  304.18
  5868.5  303.18  5878.5  304.51  5887.5  305.84  5892.9  305.19  5993.5  307.97
#Mann= 9 ,-1 , 0
  3767.8     .05       0  4150.9     .16       0  4719.7     .12       0
  4989.3     .07       0  4995.3     .12       0  5086.3     .05       0
  5560.6      .1       0  5669.5     .07       0  5878.5     .05       0
Bank Sta=4962.6,5046.4
XS Rating Curve= 0 ,0
Exp/Cntr=0.3,0.1

Type RM Length L Ch R = 1 ,99850   ,1369,1369,1369
BEGIN DESCRIPTION:
CARTERS CREEK 52.0
END DESCRIPTION:
XS GIS Cut Line= 4
      3553846.54     10237901.36      3553132.99     10237245.76
      3552882.85     10236828.65      3551897.79     10236321.53
#Sta/Elev= 30
  3623.1  306.03  3722.2  305.95  3868.1  305.47  3947.2  302.81  4001.1  299.73
  4036.5  301.98  4088.9  299.69  4114.1  299.32  4239.7  297.74  4485.3  294.68
  4543.7   294.5  4667.6  294.37  4974.4  293.48    4990  290.13  4992.8  286.61
  4995.5  286.11  4998.8  286.61    5005  286.86  5017.2  292.81    5040  295.21
  5087.4  296.16    5203  299.68    5363  299.32  5754.1  300.28  5795.4  295.57
    5903  300.49  6011.9  302.54  6027.8  302.96  6120.7  306.06  6186.4  306.75
#Mann= 19 ,-1 , 0
  3623.1     .05       0  3722.2     .16       0  3868.1     .05       0
  3947.2     .08       0  4088.9     .05       0  4114.1     .08       0
  4239.7     .05       0  4485.3     .12       0  4543.7     .16       0
  4667.6     .12       0  4992.8     .07       0  4998.8     .12       0
  5087.4     .05       0    5363     .16       0  5795.4      .1       0
    5903     .16       0  6011.9     .05       0  6027.8      .1       0
  6120.7     .05       0
#XS Ineff= 1 ,-1
 5415.91  6012.5  300.89
Permanent Ineff=
       F
Bank Sta=4974.4,5040
XS Rating Curve= 0 ,0
Exp/Cntr=0.3,0.1

Type RM Length L Ch R = 1 ,98481   ,1039,1039,1039
BEGIN DESCRIPTION:
CARTERS CREEK 51.0
END DESCRIPTION:
XS GIS Cut Line= 4
      3554653.87     10237015.98      3553955.06     10236486.44
      3553253.29     10236436.33      3552125.28     10235949.04
#Sta/Elev= 30
    3845  310.79    3935  307.27  4162.8  303.67    4221  302.92  4248.7  299.06
  4276.6  301.41  4396.9   300.7  4428.1  300.72  4725.8  300.92  4794.9  299.03
  4859.7  300.69  4948.7  297.32  4975.4  294.12  4992.1  284.53  4994.9  284.03
  4998.1  284.53  5000.1  286.48  5005.5  284.68  5025.5  291.37  5055.6  292.11
    5236  289.62  5366.7  292.95  5742.5  293.35  5925.6  296.67  5983.5  295.03
    6007  292.69  6123.8  294.87  6211.3  293.21  6583.3  302.17  6654.1  304.07
#Mann= 10 ,-1 , 0
    3845     .16       0  4162.8     .05       0  4276.6     .08       0
  4396.9      .1       0  4428.1     .08       0  4948.7     .12       0
  4992.1     .07       0  4998.1     .12       0  5366.7     .16       0
  6583.3     .05       0
#XS Ineff= 1 ,-1
 5924.15 6451.14  296.86
Permanent Ineff=
       F
Bank Sta=4975.4,5055.6
XS Rating Curve= 0 ,0
Exp/Cntr=0.3,0.1

Type RM Length L Ch R = 1 ,97442   ,1382,1382,1382
BEGIN DESCRIPTION:
CARTERS CREEK 49.0
END DESCRIPTION:
XS GIS Cut Line= 3
       3554896.9     10236230.37      3553185.09     10235699.55
      3552409.89     10235553.28
#Sta/Elev= 30
  3590.8  307.03  3856.7  304.64  4043.5  299.41  4085.6  299.43  4171.7  295.59
  4354.9  294.87  4380.8  295.88  4421.4  296.97  4604.1   296.1  4746.8  294.63
  4882.4  289.23  4964.5  290.42  4977.8  290.44  4985.4  287.24  4990.6  287.08
  4995.8  283.32  4998.5  282.82  5001.8  283.32  5009.2  285.24    5018  290.92
  5223.9  290.87  5281.4  290.25  5302.4  287.94  5336.8  288.44  5359.5  287.87
    5679  299.28  5719.5  298.18  5966.1  303.78    6137  303.52  6171.9  304.08
#Mann= 14 ,-1 , 0
  3590.8     .08       0  3856.7      .1       0  4043.5     .08       0
  4085.6      .1       0  4354.9     .08       0  4380.8      .1       0
  4421.4     .08       0  4604.1     .05       0  4964.5     .12       0
  4995.8     .07       0  5001.8     .12       0  5336.8     .05       0
    5679     .08       0    6137      .1       0
Bank Sta=4977.8,5018
XS Rating Curve= 0 ,0
Exp/Cntr=0.3,0.1

Type RM Length L Ch R = 1 ,96060   ,178,178,178
BEGIN DESCRIPTION:
CARTERS CREEK 47.1
END DESCRIPTION:
XS GIS Cut Line= 4
      3554736.36     10235902.84       3553946.4     10235128.08
      3553438.59     10234785.19       3552939.5     10234750.47
#Sta/Elev= 30
  3353.9  304.01  3428.5  304.07    3570  300.67  3605.3  298.06  3750.5  297.89
  3780.2  296.45  3883.6  296.59  3926.4  296.64  3994.1   294.4  4072.6  295.67
    4283  293.62    4365  293.25  4416.1  292.69  4597.8  287.86  4716.3  288.41
  4791.3  287.74    4806  285.86  4943.8  285.93  4964.8  280.71  5012.7  280.27
  5015.5  279.77  5018.7  280.27  5047.6  282.34  5066.7     288  5099.7  294.41
  5149.8  294.67    5230  301.56  5337.8  305.24  5487.5  304.79  5573.4   303.8
#Mann= 15 ,-1 , 0
  3353.9      .1       0  3750.5     .08       0  3780.2     .05       0
  3883.6     .08       0  3926.4      .1       0  4072.6     .08       0
    4283     .05       0    4365     .08       0  4416.1     .12       0
  4597.8     .08       0  4716.3     .12       0  5012.7     .07       0
  5018.7     .12       0  5047.6     .05       0  5487.5     .08       0
Bank Sta=4943.8,5066.7
XS Rating Curve= 0 ,0
Exp/Cntr=0.3,0.1

Type RM Length L Ch R = 1 ,95882   ,879,879,879
BEGIN DESCRIPTION:
CARTERS CREEK 47.0
END DESCRIPTION:
XS GIS Cut Line= 4
      3554857.83      10235785.6      3553989.81     10234943.61
      3553481.99     10234600.73      3552982.84     10234566.01
#Sta/Elev= 30
  3328.9  303.92  3428.1  301.69  3482.9  300.81  3575.2  298.31  3615.3  299.08
  3722.3  297.74  3742.7  297.54  3922.7  295.66  4077.1  293.71  4145.2  294.61
  4163.5  294.93  4277.7  294.52  4457.7  292.81  4567.1  286.78    4618  288.42
  4767.9  286.42  4833.8  289.77  4905.8  288.49  4933.6  287.31  4956.7  281.32
  5025.6  280.41  5028.4  279.91  5031.6  280.41  5047.3  283.45  5064.6  288.88
  5070.6  287.17  5106.6  292.27  5150.4  294.35  5422.7  301.37  5651.3  301.14
#Mann= 18 ,-1 , 0
  3328.9      .1       0  3428.1     .05       0  3482.9      .1       0
  3575.2     .08       0  3615.3      .1       0  3722.3     .05       0
  3742.7     .08       0  3922.7      .1       0  4077.1     .08       0
  4145.2      .1       0  4163.5     .08       0  4277.7      .1       0
  4457.7     .08       0  5025.6     .07       0  5031.6     .08       0
  5047.3     .05       0  5150.4     .08       0  5422.7      .1       0
Bank Sta=4905.8,5064.6
XS Rating Curve= 0 ,0
Exp/Cntr=0.3,0.1

Type RM Length L Ch R = 1 ,95003   ,1884,1884,1884
BEGIN DESCRIPTION:
CARTERS CREEK 46.0
END DESCRIPTION:
XS GIS Cut Line= 3
       3555439.4     10235297.18      3553855.23     10234094.95
      3552779.05     10234451.78
#Sta/Elev= 30
  3614.5  302.96  3951.3  298.73  4059.4  298.97  4130.1     302    4199  299.42
  4209.3  299.54  4334.9  298.11  4428.6  296.28  4508.7  292.94  4594.8  292.57
  4637.6  292.68  4829.2  284.97  4893.5   284.2  4966.2  287.07  4979.5  286.86
  4998.6  281.92  5001.3  281.42  5004.6  281.92  5022.4  286.55    5037  287.24
  5186.7  285.84  5352.4  287.31  5600.6  293.58  5879.2  294.66  6022.6  295.08
  6270.5  297.38  6312.6  299.42  6481.3  299.17  6687.6  297.03    6737  299.21
#Mann= 14 ,-1 , 0
  3614.5     .05       0    4199     .08       0  4209.3      .1       0
  4334.9     .08       0  4428.6      .1       0  4594.8     .08       0
  4829.2     .12       0  4998.6     .07       0  5004.6     .12       0
  5352.4     .05       0  5879.2      .1       0  6022.6     .05       0
  6270.5      .1       0  6481.3     .08       0
Bank Sta=4966.2,5037
XS Rating Curve= 0 ,0
Exp/Cntr=0.3,0.1

Type RM Length L Ch R = 1 ,93119   ,1768,1768,1768
BEGIN DESCRIPTION:
CARTERS CREEK 45.0
END DESCRIPTION:
XS GIS Cut Line= 4
       3555418.6     10235210.41      3554887.35     10233351.03
      3554467.13     10233094.63       3553533.2      10232069.8
#Sta/Elev= 30
  2853.3  301.88  3224.8  297.67  3328.1  298.08  3362.2  297.51    3445  296.27
  3741.5  291.71  3844.9  288.11  3948.2  286.39  3963.3  285.96  4182.4  283.59
  4256.6  284.33  4944.4  284.65  4980.7  283.97  5002.5  279.31  5015.8  284.45
  5039.2  285.06  5066.4  283.31  5078.9  278.49  5081.6  277.99  5084.9  278.49
  5109.5  284.94  5162.8  283.64  5437.9  286.93  5616.1  291.11  5950.3  303.36
  6304.3  310.46  6438.8   307.7  6460.4  311.17  6532.4  312.08  6665.9  311.62
#Mann= 17 ,-1 , 0
  2853.3     .05       0  3224.8     .16       0  3328.1     .05       0
  3362.2     .08       0    3445      .1       0  3741.5     .08       0
  3844.9     .05       0  3948.2     .16       0  3963.3      .1       0
  4182.4     .16       0  4256.6     .12       0  5078.9     .07       0
  5084.9     .12       0  5162.8     .05       0  5437.9     .08       0
  5616.1      .1       0  6532.4     .05       0
Bank Sta=5039.2,5109.5
XS Rating Curve= 0 ,0
Exp/Cntr=0.3,0.1

Type RM Length L Ch R = 1 ,91351   ,939,939,939
BEGIN DESCRIPTION:
CARTERS CREEK 44.0
END DESCRIPTION:
XS GIS Cut Line= 5
      3557402.95      10234720.8      3556142.56     10233798.94
      3555679.02     10233449.99      3555662.19     10232901.08
      3553842.08     10231391.62
#Sta/Elev= 30
    2570  313.12    2750  307.97  2868.9   305.6  3026.3  301.59  3420.8  292.58
    3750  292.48  4120.6   283.1  4296.5  282.63  4407.6  282.71  4436.7  277.27
  4457.5  282.47  4920.2  282.42  4970.2  280.45  4997.2  273.49    5000  272.99
  5003.2  273.49  5030.2  282.85  5063.3  282.75  5277.7  282.81  5762.4  285.84
  6038.6   286.1  6151.7  286.08  6292.1  288.74  6441.9  290.68  6714.1  295.16
  6981.8  301.33  7236.3  310.04  7363.1   311.6  7415.6  315.98  7625.5  322.16
#Mann= 20 ,-1 , 0
    2570     .08       0    2750     .05       0  2868.9      .1       0
  3026.3     .05       0  3420.8      .1       0  4120.6      .1       0
  4296.5     .12       0  4997.2     .07       0  5003.2     .12       0
  5063.3     .16       0  5277.7     .05       0  5762.4     .08       0
  6038.6     .05       0  6151.7     .08       0  6292.1      .1       0
  6441.9     .08       0  6714.1      .1       0  6981.8     .08       0
  7236.3      .1       0  7415.6     .08       0
#XS Ineff= 1 ,-1
 5934.09  6312.5  287.05
Permanent Ineff=
       F
Bank Sta=4920.2,5030.2
XS Rating Curve= 0 ,0
Exp/Cntr=0.3,0.1

Type RM Length L Ch R = 1 ,90412   ,768,768,768
BEGIN DESCRIPTION:
CARTERS CREEK 43.0
END DESCRIPTION:
XS GIS Cut Line= 3
      3557540.14     10234505.55      3555878.74     10232674.93
      3554692.93     10231331.95
#Sta/Elev= 30
  2843.5   310.2  2934.4  309.22  3107.1  306.94  3134.9  306.54  3156.6  303.85
    3241   304.7  3531.6  298.85  4083.7  294.43  4564.9  280.95  4736.5  281.48
  4772.5  279.77  4947.4  281.35  4975.8  279.94  4993.7   272.7  4996.5   272.2
  4999.7   272.7  5025.1  281.83    5167  279.29  5352.5  279.79  5535.8  283.28
  5903.8  282.66  5990.6  285.26  6087.9   283.4  6279.4  286.67  6392.3   290.1
    6568  298.91  6891.4  311.14    6923   311.4  7065.8  312.93  7107.2  313.19
#Mann= 14 ,-1 , 0
  2843.5     .08       0  2934.4     .05       0  3107.1      .1       0
  4736.5     .16       0  4772.5     .12       0  4993.7     .07       0
  4999.7     .12       0  5352.5     .16       0  5535.8     .05       0
  5990.6     .08       0    6568      .1       0  6891.4     .08       0
    6923     .05       0  7065.8     .08       0
#XS Ineff= 1 ,-1
 6019.32 6363.64  285.64
Permanent Ineff=
       F
Bank Sta=4947.4,5025.1
XS Rating Curve= 0 ,0
Exp/Cntr=0.3,0.1

Type RM Length L Ch R = 1 ,89644   ,1811,1811,1811
BEGIN DESCRIPTION:
CARTERS CREEK 40.0
END DESCRIPTION:
XS GIS Cut Line= 3
      3557852.63     10234297.21      3556519.29     10232269.43
       3555142.1     10231241.64
#Sta/Elev= 30
    2766  302.56  3120.9  298.46  3977.9   293.7  4250.5  290.35    4495  282.11
  4806.1  279.36  4943.4  279.98  4979.6  278.91  4997.7  271.57  5000.4  271.07
  5003.7  271.57  5009.8   271.7  5022.7  278.32  5051.9  276.06  5067.4  279.32
  5103.1  282.29  5181.4  280.51  5252.8  283.99    5282  283.49  5296.6  280.44
  5475.9  277.05  5761.5   281.6  6138.9  282.38    6280  286.38  6403.6  288.15
  6432.8  291.57    6579  297.41  6618.5  298.93  6753.9   304.2  6911.3  308.29
#Mann= 12 ,-1 , 0
    2766     .08       0  3120.9      .1       0  3977.9     .05       0
    4495     .16       0  4806.1     .12       0  4997.7     .07       0
  5003.7     .12       0  5067.4     .05       0    6280     .08       0
    6579      .1       0  6618.5     .08       0  6753.9      .1       0
Bank Sta=4943.4,5103.1
XS Rating Curve= 0 ,0
Exp/Cntr=0.3,0.1

Type RM Length L Ch R = 1 ,87833   ,1529,1529,1529
BEGIN DESCRIPTION:
CARTERS CREEK 39.0
END DESCRIPTION:
XS GIS Cut Line= 4
      3559505.36     10232665.26      3558442.91     10232595.82
      3557206.79     10231324.99      3555409.42      10230506.1
#Sta/Elev= 30
  2344.8   312.6  2395.2   312.1  2540.8  309.85  2618.6  307.82  2678.8  311.44
  2814.7  311.83  3000.8   313.4  3413.7  312.27  3708.5  306.32  3905.1  300.03
  4252.9  289.62  4430.3  287.24  4646.7  281.77  4940.5  278.35  4968.8  276.88
  5001.3  268.32    5004  267.82  5007.3  268.32  5039.5  278.91  5283.1  278.41
  5462.2  280.24  5626.7  289.43  5950.7  298.09  6159.6  297.05    6306  292.81
  6585.9  298.61  6799.1  301.69  6905.6  301.98  7084.4  304.92  7157.5  307.27
#Mann= 20 ,-1 , 0
  2344.8     .16       0  2395.2     .05       0  2540.8     .08       0
  2814.7     .05       0  3000.8     .05       0  3708.5     .08       0
  3905.1     .05       0  4252.9     .08       0  4430.3     .16       0
  4646.7     .12       0  5001.3     .07       0  5007.3     .12       0
  5283.1     .05       0  5626.7      .1       0  6159.6     .08       0
    6306      .1       0  6585.9     .05       0  6799.1     .08       0
  6905.6     .05       0  7084.4      .1       0
Bank Sta=4940.5,5039.5
XS Rating Curve= 0 ,0
Exp/Cntr=0.3,0.1

Type RM Length L Ch R = 1 ,86304   ,257,257,257
BEGIN DESCRIPTION:
CARTERS CREEK 37.0
END DESCRIPTION:
XS GIS Cut Line= 3
      3559788.96     10231350.83      3558532.02     10230621.67
      3555781.98     10230503.61
#Sta/Elev= 30
  2849.8  319.78  2941.1  311.47  3577.2   292.4    3721  291.13  3936.5  283.56
  3989.5  286.26    4421  281.05  4573.1  283.31  4633.1  278.04  4728.2  277.03
  4857.9  276.04  4943.4  278.28  4963.4  276.25  4980.5  268.89  4983.2  268.39
  4986.5  268.89  5003.5   268.9  5043.5  277.62  5217.2  278.54  5320.1  278.77
  5517.4  287.15  5714.7  289.02  5764.2  288.16  5804.2   281.8  5830.4  285.26
  5939.2  291.75  6104.5  292.91  6204.6  298.09  6609.9     298  7055.5  303.75
#Mann= 15 ,-1 , 0
  2849.8     .05       0  3577.2      .1       0    3721     .05       0
    4421     .08       0  4728.2      .1       0  4857.9     .12       0
  4980.5     .07       0  4986.5     .12       0  5217.2      .1       0
  5320.1     .05       0  5517.4     .08       0  5714.7     .16       0
  5830.4     .08       0  5939.2      .1       0  6609.9     .05       0
#XS Ineff= 1 ,-1
 4154.55 4567.05  283.43
Permanent Ineff=
       F
Bank Sta=4943.4,5043.5
XS Rating Curve= 0 ,0
Exp/Cntr=0.3,0.1

Type RM Length L Ch R = 1 ,86047   ,764,764,764
BEGIN DESCRIPTION:
CARTERS CREEK 36.0
END DESCRIPTION:
XS GIS Cut Line= 5
      3560080.68     10230663.35      3558920.91     10230232.78
      3558379.24      10230392.5      3557733.41     10230343.89
      3555748.46     10230276.38
#Sta/Elev= 30
  2743.1  307.14  2869.6   308.9  2926.6  308.18  3159.6   305.6  3317.6  292.42
  3388.3  292.18    3990  278.35  4094.1  279.42  4125.4  279.48  4302.4  278.16
  4406.6  279.88  4667.5  282.44  4712.5  276.78  4963.3  277.73  5000.4  267.53
  5003.1  267.03  5006.4  267.53  5033.5  277.95    5314  269.61    5354  281.32
  5684.2  291.83  5885.6  291.04  5944.3  285.59  5974.4  291.89  6117.9  295.34
  6802.3  299.94  6874.4  300.25  6979.3   302.9  7176.6  307.35  7178.7  307.35
#Mann= 19 ,-1 , 0
  2743.1     .08       0  2869.6      .1       0  2926.6     .08       0
  3159.6     .05       0  3388.3      .1       0    3990     .08       0
  4094.1      .1       0  4125.4     .08       0  4302.4      .1       0
  4406.6     .15       0  4667.5      .1       0  5000.4     .07       0
  5006.4      .1       0  5885.6     .08       0  6117.9      .1       0
  6802.3     .08       0  6874.4      .1       0  6979.3     .15       0
  7176.6     .08       0
#XS Ineff= 1 ,-1
 3343.18 4601.14  283.72
Permanent Ineff=
       F
Bank Sta=4963.3,5033.5
XS Rating Curve= 0 ,0
Exp/Cntr=0.3,0.1

Type RM Length L Ch R = 1 ,85283   ,363,363,363
BEGIN DESCRIPTION:
CARTERS CREEK 34.1
END DESCRIPTION:
XS GIS Cut Line= 4
      3559879.21     10230218.88      3558018.13     10229684.17
      3557587.58       10229330.       3556727.6     10229012.48
#Sta/Elev= 30
  2937.9  304.27  3018.6  302.11  3377.1  282.09  3526.5  277.74  3569.6  282.45
    3628  281.68  3762.8  274.15  3902.5  274.51  3944.1   280.5  4135.9  280.78
  4440.6  281.45  4526.8  280.84  4559.8  276.49  4647.2  283.55  4745.3  285.46
  4846.9  281.59    4916  275.12  4951.2  277.14    5012  267.29  5014.8  266.79
    5018  267.29  5088.6  271.65  5136.3  276.79  5212.4  280.58  5468.1  281.92
  5728.5   285.4  5870.4  288.64  6077.8  292.65  6293.4  294.98  6348.5  296.73
#Mann= 20 ,-1 , 0
  2937.9     .16       0  3018.6      .1       0  3377.1     .05       0
  3526.5     .08       0    3628      .1       0  3762.8      .1       0
  4135.9     .12       0  4440.6      .1       0  4559.8      .1       0
  4745.3     .08       0  4846.9     .12       0    5012     .07       0
    5018     .12       0  5088.6     .12       0  5212.4     .16       0
  5468.1     .08       0  5728.5     .08       0  5870.4      .1       0
  6077.8      .1       0  6293.4     .15       0
#XS Ineff= 1 ,-1
 3115.91 4734.09  286.03
Permanent Ineff=
       F
Bank Sta=4951.2,5136.3
XS Rating Curve= 0 ,0
Exp/Cntr=0.3,0.1
