HEC-RAS study GIBBONS CREEK.prj: GIBBONS CREEK Base Level Engineering

--- GIBBONS CREEK.g01 (geometry) --- (continued)

Type RM Length L Ch R = 1 ,83018   ,1769,1769,1769
BEGIN DESCRIPTION:
GIBBONS CREEK 58.0
END DESCRIPTION:
XS GIS Cut Line= 4
      3646642.13     10221891.63       3645333.3     10222415.16
      3644494.92     10223478.94      3644850.82     10225171.64
#Sta/Elev= 30
  2917.9  272.29  3004.1  269.31  3154.9  261.09  3243.3  259.05  3285.5  259.27
  3333.9  261.61  3358.2  261.65  3434.9  258.14  3632.8   255.4  3693.4  252.82
  3831.6  249.11  3862.7     247  3865.5   246.5  3868.7     247  6531.4     247
  6632.6   247.4  6762.3  249.92  6807.1   252.3  6822.7  251.99  6835.1  252.56
  6839.5  252.77  6856.9  254.12    6862  253.35  6906.8  255.12  6972.3  254.56
  7067.3   257.2  7186.9  262.66  7250.6  262.55  7360.6  265.13  7411.7  264.15
#Mann= 10 ,-1 , 0
  2917.9     .05       0  3243.3     .16       0  3831.6     .05       0
  3862.7    .033       0  3868.7     .05       0  6531.4     .16       0
  6632.6     .05       0  6822.7     .16       0  6835.1     .05       0
  7067.3     .16       0
Bank Sta=3693.4,6839.5
XS Rating Curve= 0 ,0
Exp/Cntr=0.3,0.1

Type RM Length L Ch R = 1 ,81249   ,4761,4761,4761
BEGIN DESCRIPTION:
GIBBONS CREEK 57.0
END DESCRIPTION:
XS GIS Cut Line= 4
      3646632.92      10221187.1      3644382.07     10221176.42
      3642867.41     10222294.68      3641029.22     10223932.49
#Sta/Elev= 30
  1808.3  269.31  1948.6  268.82  2029.1  268.65  2129.1  266.26  2589.1  264.79
  2679.1  262.96  2909.1  253.79  2969.1  253.82  2989.1  252.49  3029.1  251.27
  3089.1  252.55  3189.1  251.89  3309.1  247.17  3356.1  246.82  3358.9  246.32
  3362.1  246.82  3380.8     247    6900     247    7013  253.06  7225.3  267.63
  7466.1     272  7643.4     278  7698.4  277.72  7728.7  275.33    7778  273.89
  7933.5  271.97  8104.1  273.25  8164.9  270.22    8177  269.44  8403.9  273.18
#Mann= 8 ,-1 , 0
  1808.3     .05       0  1948.6     .16       0  3356.1    .033       0
  3362.1     .16       0  3380.8     .05       0  7698.4     .16       0
  8164.9     .05       0    8177     .16       0
Bank Sta=2989.1,7013
XS Rating Curve= 0 ,0
Exp/Cntr=0.3,0.1

Type RM Length L Ch R = 1 ,76460   ,1067,1067,1067
BEGIN DESCRIPTION:
GIBBONS CREEK 55.0
END DESCRIPTION:
XS GIS Cut Line= 3
      3646232.05     10217414.62      3639898.75     10218269.28
      3633201.43     10217046.72
#Sta/Elev= 30
  -705.8  251.41  -362.8  257.31  -214.8  253.67  -191.2  253.02     -67  248.81
   -42.9     247   -40.1   246.5   -36.9     247 10817.1     247 10922.4     247
 10957.3  249.86 10967.4  255.64 10977.6  260.13 10986.2  260.98 11028.4  261.23
 11038.6  260.02 11044.6   257.6 11049.6  257.85 11058.9   254.8 11066.3  249.72
 11069.1   247.8   11305  247.31   11515  257.81 11575.5  262.36 11628.2  265.26
 11820.6  266.72 12143.3  275.33 12245.6  276.13 12279.1   276.3 12492.9  276.73
#Mann= 14 ,-1 , 0
  -705.8     .05       0  -214.8     .16       0     -67     .05       0
   -42.9    .033       0   -36.9     .05       0 10817.1     .07       0
 10922.4     .15       0 11066.3     .05       0   11305     .16       0
   11515     .05       0 11575.5     .16       0 12143.3      .1       0
 12245.6     .16       0 12279.1      .1       0
#XS Ineff= 1 ,-1
 -736.36 -354.55  257.44
Permanent Ineff=
       F
Bank Sta=-191.2,10967.4
XS Rating Curve= 0 ,0
Exp/Cntr=0.3,0.1

Type RM Length L Ch R = 1 ,75421   ,1052,1052,1052
BEGIN DESCRIPTION:
GIBBONS CREEK 52.0
END DESCRIPTION:
XS GIS Cut Line= 3
      3645048.68     10216790.57      3639069.81     10217253.13
      3633995.29     10215951.25
#Sta/Elev= 30
   188.5  262.18   315.5  262.13   487.3  254.68   586.3  249.88   596.3     247
    1830     247  1930.3  250.39  2007.5  246.85  2010.3  246.35  2013.5  246.85
  2953.3     247  2963.3  251.17  2994.1  254.84  3053.6   255.7  3119.1  251.95
  3153.9  250.67  3163.9     247 10118.1  246.89 10570.5  253.17 10601.4  253.57
 10637.7   251.7 10684.1  254.58 10714.1  260.61 10795.6  262.11 10828.6  255.22
 10873.4  254.62 10963.9  261.79 11279.7  263.37 11320.5  270.21 11424.1   271.1
#Mann= 6 ,-1 , 0
   188.5     .16       0   487.3     .05       0  2007.5    .033       0
  2013.5     .05       0 10601.4      .1       0 10873.4     .08       0
Bank Sta=3119.1,10570.5
XS Rating Curve= 0 ,0
Exp/Cntr=0.3,0.1

Type RM Length L Ch R = 1 ,74369   ,1682,1682,1682
BEGIN DESCRIPTION:
GIBBONS CREEK 50.0
END DESCRIPTION:
XS GIS Cut Line= 3
      3644880.92     10215861.75      3638798.65     10216228.07
      3635192.06     10215491.63
#Sta/Elev= 30
    40.2  259.12   122.9  259.76   259.4  256.61     557  246.87   559.7  246.37
     563  246.87   770.3   255.1   954.5  259.61  1158.4   266.9  1209.8   268.4
  1261.2  268.88  1286.1  271.28  1321.3  269.16  1454.4  268.77  1651.9   265.4
  1742.1  262.91  1986.6  249.19  2022.6     247  8997.9     247  9093.5     249
  9212.3  252.89  9300.1  255.83  9324.5     258  9375.6  256.75  9390.2   257.5
    9396  259.63  9406.2  260.41  9457.2   260.3  9620.5  266.75  9814.5  272.14
#Mann= 8 ,-1 , 0
    40.2     .16       0     557    .033       0     563     .16       0
  1158.4      .1       0  1209.8     .16       0  1986.6     .05       0
  9093.5     .16       0  9300.1     .05       0
Bank Sta=557,9212.3
XS Rating Curve= 0 ,0
Exp/Cntr=0.3,0.1

Type RM Length L Ch R = 1 ,72687   ,3321,3321,3321
XS GIS Cut Line= 2
     3643376.273    10215874.474     3634876.273    10213103.641
#Sta/Elev= 30
       0  267.31  109.88  264.22  289.68  253.47  329.64  254.64  379.58     247
 7381.86     247 7411.82  251.38 7451.78  248.83 7481.75  255.29  7521.7  264.06
 7631.58  271.36 7681.53  280.46 7761.44  283.49 7811.38  281.52 7861.33  272.01
  7891.3  262.67 7901.28  261.92 7941.24  265.55 7971.21  262.35 8001.17  269.83
 8041.13  273.85  8071.1  272.04 8200.95  272.03 8240.91  268.11 8480.65   270.3
 8510.61  267.82 8760.34   270.6  8790.3  269.02 8830.26  270.88  8880.2  269.19
#Mann= 5 ,-1 , 0
       0     .16       0  329.64    .033       0 7411.82     .08       0
 7761.44     .05       0 8041.13      .1       0
Bank Sta=329.64,7481.75
XS Rating Curve= 0 ,0
Exp/Cntr=0.3,0.1

Type RM Length L Ch R = 1 ,69366   ,195,195,195
BEGIN DESCRIPTION:
GIBBONS CREEK 46.1
END DESCRIPTION:
XS GIS Cut Line= 5
     3643376.273    10215770.308      3641730.44    10213207.808
     3639126.273    10211436.974     3637938.773    10211059.646
     3635188.773    10211707.808
#Sta/Elev= 30
  1233.9  253.61    1283  261.02  1363.3  253.07  1584.1     247  4583.9     247
  4691.6     247  5287.2  246.83  5293.2  246.83  5314.7  247.11  5597.3   253.4
  5904.4  254.99  6034.9   250.8  6344.3  247.61  6498.2  260.98  6807.9  258.38
  7411.4  264.42  7575.6  255.63  8059.3  274.99    8145  285.43  8192.9  284.37
  8355.3  284.88  8460.4  263.24  8551.3  263.52    8685  285.46    8809   284.1
    8809251.35539497.212234.700510145.53236.678911093.06257.142411192.81263.5099
#Mann= 8 ,-1 , 0
  1233.9     .05       0  4583.9     .08       0  4691.6     .05       0
  5287.2    .033       0  5293.2     .05       0  5314.7     .08       0
  6034.9     .05       0  8192.9     .08       0
#XS Ineff= 2 ,-1
  1187.5 1289.77  261.46 8713.6411222.73   286.7
Permanent Ineff=
       F       F
Bank Sta=1363.3,5597.3
XS Rating Curve= 0 ,0
Exp/Cntr=0.3,0.1

Type RM Length L Ch R = 1 ,69171   ,143,143,143
BEGIN DESCRIPTION:
GIBBONS CREEK 46.0
END DESCRIPTION:
XS GIS Cut Line= 6
     3643813.773    10215249.474     3642459.606    10214061.974
     3641709.606    10212916.141     3639188.773    10211311.974
     3638063.773    10210895.308     3635251.273    10211541.141
#Sta/Elev= 30
    1334  250.89  1585.1  247.16  1681.6  259.48  1798.8  260.92  4444.9  255.35
    4502  250.57  4640.1  259.49  4889.3  259.86  4894.8  259.86  4909.4  259.87
  4928.5  245.65  4930.8  236.28  4936.8  236.28    4991  245.32  5027.5  241.73
  5058.8   256.6  5174.1  258.93  5454.3  260.33    5673  251.17    6091  260.74
  6497.3  255.12  7043.1  263.35  7728.5  260.21  8017.6  267.96  8631.4  283.65
  8745.1  264.928754.998250.55369304.877233.103910384.64244.935611174.46266.8802
#Mann= 8 ,-1 , 0
    1334     .05       0  4889.3     .08       0  4894.8     .05       0
  4930.8    .033       0  4936.8     .05       0  5174.1     .08       0
  7043.1     .05       0  8017.6     .08       0
#XS Ineff= 1 ,-1
 8631.8211113.64  283.24
Permanent Ineff=
       F
Bank Sta=4909.4,5058.8
XS Rating Curve= 0 ,0
Exp/Cntr=0.3,0.1

Type RM Length L Ch R = 1 ,69028   ,401,401,401
BEGIN DESCRIPTION:
GIBBONS CREEK 45.0
END DESCRIPTION:
XS GIS Cut Line= 5
     3644397.106    10214332.808     3641938.773    10212728.641
      3639276.83      10211144.7      3638157.08     10210759.65
      3635345.81     10211405.21
#Sta/Elev= 30
  -935.4  264.38  -668.8  267.64    -590  264.79  -210.8   253.5  -111.7  251.78
   482.9  239.93     582  236.58   802.4  232.61  1077.5  230.94  1176.6  233.59
  1372.7  238.84  1374.8   238.9  1547.6  243.37  2285.1  225.22  4125.3  222.86
    4156  215.72  4236.8  224.65  4683.6  248.27  4782.6  222.85  4930.5  214.87
  4933.2  214.37  4936.5  214.87  5037.4  215.56  5178.1  224.93  5279.1  244.95
  5823.5  252.92  6051.8  253.57  7141.4  262.26  8109.2  273.54  8729.3  283.88
#Mann= 19 ,-1 , 0
  -935.4      .1       0  -668.8     .16       0    -590      .1       0
  -210.8     .05       0  -111.7     .16       0   482.9     .05       0
     582     .12       0   802.4     .16       0  1077.5     .12       0
  1176.6     .05       0  1372.7      .1       0  1374.8     .05       0
  4930.5    .033       0  4936.5     .05       0  5037.4     .08       0
  5823.5     .05       0  6051.8     .08       0  7141.4     .05       0
  8109.2     .08       0
#XS Ineff= 1 ,-1
    4675 5370.45  248.45
Permanent Ineff=
       F
Bank Sta=2285.1,4236.8
XS Rating Curve= 0 ,0
Exp/Cntr=0.3,0.1

Type RM Length L Ch R = 1 ,68627   ,1526,1526,1526
XS GIS Cut Line= 3
        3643757.       10212359.        3638210.       10210354.
        3635407.       10211031.
#Sta/Elev= 30
       0262.5681119.6312261.4146418.7093253.43581176.374231.84062532.195222.3096
3150.289219.81723369.613219.5758 3549.06220.73193888.015221.83114007.646214.8618
4087.401223.22074147.216222.2393 4366.54218.23994705.495236.22124805.188216.2911
4845.065209.64955024.512210.81555104.266232.1498 5184.02238.77575383.406242.6532
5542.914233.38325802.115247.26676001.407248.8925 6280.33 248.0436559.252245.7866
6878.021253.50447176.866255.94987356.173254.94858691.016277.98498770.708289.2666
#Mann= 17 ,-1 , 0
       0      .1       0119.6312     .05       0418.7093      .1       0
3150.289     .05       03369.613     .16       0 3549.06     .12       0
3888.015     .07       04147.216      .1       04805.188     .05       0
 5184.02     .16       05802.115      .1       06001.407     .16       0
 6280.33      .1       06559.252     .16       06878.021      .1       0
7176.866     .16       07356.173     .08       0
#XS Ineff= 1 ,-1
 4704.55 5363.64  236.17
Permanent Ineff=
       F
Bank Sta=2532.195,4087.401
XS Rating Curve= 0 ,0
Exp/Cntr=0.3,0.1

Type RM Length L Ch R = 1 ,66881   ,2519,2519,2519
BEGIN DESCRIPTION:
GIBBONS CREEK 44.0
END DESCRIPTION:
XS GIS Cut Line= 4
      3643881.97     10209853.07      3640762.18      10209251.5
      3637715.32     10209394.74      3636027.82     10210519.73
#Sta/Elev= 30
    41.1  267.76    99.2  266.91   555.2  252.35   697.9  246.43   797.7   244.5
     921  245.83   988.1  234.16    1398  233.44    2218  219.71  2383.3  220.21
  2413.9   213.4  2450.6  220.26  4019.3  215.59  4920.3  220.48  4997.4  209.74
  5000.1  209.24  5003.4  209.74  5028.5  213.21  5040.4   220.7  5185.9  219.03
  5370.9  220.53  5568.9  222.13  6162.9  240.38  6273.5   243.3  6382.2  247.26
    7157  257.24  7454.3   256.3  8010.4  259.77  8281.6  264.33  8296.7  264.47
#Mann= 18 ,-1 , 0
    41.1      .1       0    99.2     .05       0   555.2      .1       0
   697.9     .05       0   797.7     .16       0    2218     .12       0
  4997.4     .07       0  5003.4     .12       0  5185.9      .1       0
  5370.9     .05       0  5568.9     .16       0  6162.9      .1       0
  6273.5     .16       0  6382.2      .1       0    7157     .16       0
  7454.3      .1       0  8010.4     .16       0  8281.6     .08       0
Bank Sta=4920.3,5040.4
XS Rating Curve= 0 ,0
Exp/Cntr=0.3,0.1

Type RM Length L Ch R = 1 ,64362   ,1781,1781,1781
BEGIN DESCRIPTION:
GIBBONS CREEK 42.0
END DESCRIPTION:
XS GIS Cut Line= 4
      3642992.09     10209091.64      3639958.51     10207980.15
      3638786.63     10208266.61      3636742.33     10209191.11
#Sta/Elev= 30
  1036.5  250.66  1168.4  257.16  1590.3  240.32  2058.9  233.29  2522.9  218.91
  2751.1  216.57  2921.5  224.98  3172.4  217.34  3669.7  217.86  3694.9  211.93
  3786.4   212.5  3848.1  218.33  4007.9  216.97  4039.7     212  4100.7  217.21
  4375.3  213.42  4572.4  216.48  4613.6  211.82  4644.5  217.56  4953.3  217.69
  4981.2  209.17  4983.9  208.67  4987.2  209.17    5046  216.87    5897  217.28
  6833.4  248.02  7190.7  245.23  7219.6  241.46  7346.2  248.72  7717.3  255.74
#Mann= 5 ,-1 , 0
  1036.5     .05       0  2522.9     .12       0  4981.2     .07       0
  4987.2     .12       0    5897     .16       0
Bank Sta=4953.3,5046
XS Rating Curve= 0 ,0
Exp/Cntr=0.3,0.1

Type RM Length L Ch R = 1 ,62581   ,1786,1786,1786
BEGIN DESCRIPTION:
GIBBONS CREEK 41.0
END DESCRIPTION:
XS GIS Cut Line= 4
      3643224.78     10207528.86      3639984.55     10206964.53
      3638721.31     10207269.96      3636990.64      10208357.2
#Sta/Elev= 30
   993.8  281.85  1068.8  279.25  1193.4  268.65    1492  241.98  1849.2  223.75
  2630.8  219.65  2661.2  223.16  2722.1  223.34  2810.9  218.29  2937.4  217.86
  3917.8  215.87  3940.2  213.46  4031.5  216.94    4882  216.23  4923.2   213.7
  4964.3  215.15  4992.2  207.79    4995  207.29  4998.2  207.79  5012.9  215.55
  5026.1  216.18  5727.9  215.64  6930.9  222.46  7062.5  231.66  7077.8  235.12
  7330.6  244.22  7408.9  245.13  7504.5  242.63  7528.4  241.11  7626.3  244.76
#Mann= 11 ,-1 , 0
   993.8     .05       0  1193.4     .16       0    1492     .05       0
  2937.4     .12       0  4992.2     .07       0  4998.2     .12       0
  6930.9     .16       0  7330.6      .1       0  7408.9     .16       0
  7504.5      .1       0  7528.4     .16       0
Bank Sta=4882,5026.1
XS Rating Curve= 0 ,0
Exp/Cntr=0.3,0.1

Type RM Length L Ch R = 1 ,60795   ,327,327,327
BEGIN DESCRIPTION:
GIBBONS CREEK 39.0
END DESCRIPTION:
XS GIS Cut Line= 4
      3644494.29     10206422.09      3639785.62     10205907.67
      3638350.52     10205870.55      3636519.01     10205836.15
#Sta/Elev= 30
  -405.3  272.76  -285.6  274.35  -151.6  274.86   -66.3   270.2   196.4  256.46
   763.8  239.83  1119.5  240.37    1468  234.32  1799.9  253.12    1884  252.26
  2195.8  227.16  2282.8  222.24    2494  219.91    3240  217.66  4185.5   213.1
  4580.5  212.33  4679.1  212.55    4735  212.96    4775  207.63  4822.1  207.14
  4824.8  206.64  4828.1  207.14  4935.1  215.43  4975.1  215.46  5005.1  207.24
  5035.1  214.48  6215.5  218.03  6665.5  227.96  6925.6  239.24  7598.8  244.31
#Mann= 11 ,-1 , 0
  -405.3     .05       0  -285.6     .16       0   -66.3     .05       0
    1884     .16       0  2195.8     .05       0    3240     .08       0
  4185.5     .05       0  4580.5     .08       0  4679.1     .05       0
  4822.1     .04       0  4828.1     .05       0
Bank Sta=4735,4935.1
XS Rating Curve= 0 ,0
Exp/Cntr=0.3,0.1

Type RM Length L Ch R = 1 ,60468   ,934,934,934
BEGIN DESCRIPTION:
GIBBONS CREEK 38.0
END DESCRIPTION:
XS GIS Cut Line= 4
      3643213.94     10205922.96      3639644.04     10205619.14
      3638038.14     10205543.18      3636717.05     10205547.81
#Sta/Elev= 30
   801.7  256.94   877.5  252.79   926.2  244.75  1024.3  252.78  1245.1   258.6
  1463.4     253  1646.6  258.34  1763.7  250.48  2007.9  230.95  2173.4  221.55
  2218.6  225.39  2258.8  219.75  2478.4  218.58  3670.8  215.13  3704.2  215.29
  3888.5   214.6  4859.2  215.65  4967.1  214.25  4994.1  207.45  4996.9  206.95
  5000.1  207.45  5037.2  214.98  5077.3  211.51  5117.3  215.94  6178.2  215.93
  6548.2  233.86  6918.2  243.27  7037.5  241.96  7208.2  244.19  7313.3  241.72
#Mann= 11 ,-1 , 0
   801.7     .05       0   926.2     .16       0  1763.7     .05       0
  2478.4      .1       0  3670.8     .12       0  3704.2      .1       0
  3888.5     .12       0  4859.2     .05       0  4994.1     .03       0
  5000.1     .05       0  7037.5     .08       0
Bank Sta=4967.1,5037.2
XS Rating Curve= 0 ,0
Exp/Cntr=0.3,0.1

Type RM Length L Ch R = 1 ,59534   ,3570,3570,3570
BEGIN DESCRIPTION:
GIBBONS CREEK 37.0
END DESCRIPTION:
XS GIS Cut Line= 3
      3642452.84     10205778.32      3638760.59     10204750.99
      3636992.07     10205191.65
#Sta/Elev= 30
  1640.2  257.77  1734.4  255.65    1969  238.29  2191.1  223.27  2211.9  222.62
  2245.8  226.35  2294.9  218.55  2412.1  217.09  2918.9  217.05  3000.7  214.75
  3433.3  214.35  3520.3   214.2  3710.3  214.09  3920.2  214.35  4021.5  214.32
  4122.9   214.4  4224.3  213.57  4381.2  212.39  4952.1  214.71  4967.2  213.85
  4990.7  206.07  4993.4  205.57  4996.7  206.07  5024.8  215.49  5065.6  215.69
  5800.9  213.49  6635.7  214.61  6769.7  218.47  7120.1  237.02  7295.3  239.19
#Mann= 13 ,-1 , 0
  1640.2     .16       0    1969     .05       0  2412.1      .1       0
  3433.3     .16       0  3520.3      .1       0  3710.3     .12       0
  3920.2     .05       0  4021.5      .1       0  4122.9     .05       0
  4224.3     .12       0  4990.7     .07       0  4996.7     .12       0
  5065.6     .05       0
Bank Sta=4952.1,5024.8
XS Rating Curve= 0 ,0
Exp/Cntr=0.3,0.1

Type RM Length L Ch R = 1 ,55964   ,1033,1033,1033
BEGIN DESCRIPTION:
GIBBONS CREEK 36.0
END DESCRIPTION:
XS GIS Cut Line= 3
      3641846.55     10202120.77      3638057.47     10203917.65
      3636429.86     10204269.22
#Sta/Elev= 30
  1186.7  231.06    1318  225.77  1722.9   226.5  1806.5  251.68  1822.5     253
  1844.6  249.54  1897.5   231.4  1965.7  218.38  2320.8  216.57  2848.5     215
  2880.1  213.47  2902.8   217.6  3194.8   212.7  3780.7   212.8  3817.2  211.97
  3839.9  206.97  3857.1  213.52  4965.6  212.02  4981.7  211.69  4995.8  204.74
  4998.6  204.24  5001.8  204.74  5027.2  212.35  5049.9  212.87  5096.5  212.99
  6531.6   216.4  6558.4  221.88  6715.7  221.99  6887.8  240.29  7045.4  240.93
#Mann= 7 ,-1 , 0
  1186.7     .05       0  2320.8     .12       0  2848.5     .05       0
  3780.7     .12       0  4995.8     .07       0  5001.8     .12       0
  5096.5     .05       0
Bank Sta=4965.6,5049.9
XS Rating Curve= 0 ,0
Exp/Cntr=0.3,0.1

Type RM Length L Ch R = 1 ,54931   ,1443,1443,1443
BEGIN DESCRIPTION:
GIBBONS CREEK 35.0
END DESCRIPTION:
XS GIS Cut Line= 3
      3641143.37     10200935.91      3638929.86      10202693.7
      3636892.09     10203591.65
#Sta/Elev= 30
  1790.8  234.95  1995.7  232.18  2091.5  227.42  2163.1   223.2  2316.6  215.34
  2398.6  214.75  2414.4  215.04  2694.2  214.95    3319  211.77  4029.7  211.78
  4244.2   213.7  4265.8  207.15  4286.6  211.96  4301.1  212.53  4489.9  211.08
  4540.8  211.26  4918.8   213.1  4986.5  210.18  4994.3  205.52  5005.3  203.92
  5008.1  203.42  5011.3  203.92  5023.1  206.87  5030.2  211.74    5059  212.79
  5813.3  211.05  6440.2  217.48  6562.3   220.8  6678.9  230.89  6844.2  241.63
#Mann= 13 ,-1 , 0
  1790.8     .05       0  2091.5     .12       0  2163.1     .05       0
  2316.6     .12       0  2398.6     .05       0  2414.4     .12       0
  2694.2     .05       0  4029.7     .12       0  4489.9      .1       0
  4540.8     .12       0  5005.3     .07       0  5011.3     .12       0
    5059     .05       0
Bank Sta=4918.8,5059
XS Rating Curve= 0 ,0
Exp/Cntr=0.3,0.1

Type RM Length L Ch R = 1 ,53488   ,859,859,859
BEGIN DESCRIPTION:
GIBBONS CREEK 34.0
END DESCRIPTION:
XS GIS Cut Line= 3
      3640791.82     10200245.79      3638356.94     10201834.32
      3637092.08     10202591.66
#Sta/Elev= 30
  2380.9  240.45  2876.3  217.85  3120.8  212.05  4111.9  210.02  4912.9   212.7
  4928.1   210.2  4943.2  212.41  4964.3  212.24  4979.4   210.4  4985.4  205.01
  4997.5  203.21  5000.2  202.71  5003.5  203.21  5017.7  206.21  5024.5  209.41
  5043.2  211.65    5254  210.19    5407  211.75  5523.7  209.77  5573.5  211.76
  5836.7  210.17  5879.5  211.45  5953.4  208.99  6208.2  210.17  6250.9  207.63
  6346.2   214.2  6425.9  222.36  6515.4  226.84  6558.2  231.15  6762.4  238.04
#Mann= 5 ,-1 , 0
  2380.9     .05       0  4997.5     .03       0  5003.5     .05       0
  5017.7     .12       0  5024.5     .05       0
Bank Sta=4964.3,5043.2
XS Rating Curve= 0 ,0
Exp/Cntr=0.3,0.1

Type RM Length L Ch R = 1 ,52629   ,1600,1600,1600
BEGIN DESCRIPTION:
GIBBONS CREEK 33.0
END DESCRIPTION:
XS GIS Cut Line= 3
      3640392.12     10199791.64      3638916.58     10200381.85
       3636792.1     10202391.64
#Sta/Elev= 30
  2668.6  241.87  2865.7  231.14  2911.4  228.72  3030.8  221.43  3060.4  223.39
  3084.6  219.44    3226  218.37  3378.8  216.04  3559.4  215.47    3922  213.95
  3966.6   210.9  4675.8  211.08  4968.1  211.55  5000.7  201.57  5003.4  201.07
  5006.7  201.57    5043  211.18  5046.1  211.34  5231.5  210.58  6000.9  211.85
  6073.9  207.29  6167.5  211.95  6510.2  212.02  6731.9  218.91  6760.5  219.94
    6873   224.2  6897.8  225.19  7014.1  230.25  7035.1   231.6  7182.3   235.7
#Mann= 20 ,-1 , 0
  2668.6     .05       0  2865.7     .08       0  2911.4     .05       0
    3226     .08       0  3378.8     .05       0  3559.4     .08       0
  3966.6     .05       0  4675.8     .08       0  5000.7     .07       0
  5006.7     .08       0    5043     .12       0  5231.5     .08       0
  6073.9     .05       0  6167.5     .08       0  6731.9     .05       0
  6760.5     .08       0    6873     .05       0  6897.8     .08       0
  7014.1     .05       0  7035.1     .08       0
Bank Sta=4968.1,5046.1
XS Rating Curve= 0 ,0
Exp/Cntr=0.3,0.1

Type RM Length L Ch R = 1 ,51029   ,1483,1483,1483
BEGIN DESCRIPTION:
GIBBONS CREEK 32.0
END DESCRIPTION:
XS GIS Cut Line= 3
      3640292.12     10197491.63      3637827.56     10200327.83
      3636338.73     10201925.45
#Sta/Elev= 30
  2159.5  295.72  2365.1  272.69  2457.2   258.3  2620.5  250.79    2762  236.96
  3024.1   220.1  3313.7  211.11  3441.6  208.35  3551.7  207.42  4041.5  207.07
  4849.9  209.08  4959.3   210.2  4981.2   208.8    4999  200.88  5001.8  200.38
    5005  200.88  5030.5  209.67  5506.4  208.66  5903.3  208.53  6231.8  207.64
  6599.6  209.26    6607   209.3  6966.8  211.46  7055.7  208.05  7194.7  210.66
  7437.8  209.59    7558  221.14  7635.6  233.63  7826.7  237.33  8100.7  233.33
#Mann= 15 ,-1 , 0
  2159.5     .05       0  3313.7     .16       0  3441.6     .05       0
  3551.7     .12       0  4041.5     .05       0  4849.9     .12       0
    4999     .07       0    5005     .12       0  5506.4     .05       0
  5903.3     .12       0  6231.8     .07       0  6599.6     .12       0
    6607     .05       0  6966.8     .12       0  7194.7     .05       0
Bank Sta=4959.3,5030.5
XS Rating Curve= 0 ,0
Exp/Cntr=0.3,0.1

Type RM Length L Ch R = 1 ,49546   ,5141,5141,5141
BEGIN DESCRIPTION:
GIBBONS CREEK 31.0
END DESCRIPTION:
XS GIS Cut Line= 4
      3640244.99     10197042.64      3638343.92     10198592.13
       3636895.7     10198772.03      3634841.32     10200154.63
#Sta/Elev= 30
  1972.8  296.55  2060.9  288.75  2071.9  287.18  2322.9  252.95  2378.9  252.25
  2500.2  233.43    2585  230.24  2642.4  219.83    3269  208.99  3376.2  208.76
  3417.4  208.54  3714.3  206.63  4627.7  208.37  4727.6  208.88  4961.3  208.98
  4998.6  199.61  5001.3  199.11  5004.6  199.61    5062  209.59  5730.3  207.04
  6184.6   207.3  6350.9  207.79  6468.1  208.15  6791.9  209.95    6850  210.56
  7025.5  210.88  7376.6  214.62  7709.2  233.87  7876.4  237.38    8361  232.33
#Mann= 19 ,-1 , 0
  1972.8     .05       0  2060.9     .08       0  2071.9     .05       0
    3269     .16       0  3376.2      .1       0  3417.4     .16       0
  3714.3     .12       0  4627.7     .05       0  4727.6     .12       0
  4998.6     .07       0  5004.6     .12       0  5730.3     .05       0
  6184.6     .12       0  6350.9     .16       0  6468.1     .05       0
  6791.9     .12       0    6850     .05       0  7025.5     .12       0
  7376.6     .05       0
Bank Sta=4961.3,5062
XS Rating Curve= 0 ,0
Exp/Cntr=0.3,0.1

Type RM Length L Ch R = 1 ,44405   ,2673,2673,2673
BEGIN DESCRIPTION:
GIBBONS CREEK 29.0
END DESCRIPTION:
XS GIS Cut Line= 4
       3639792.1     10196341.64      3638553.91     10197021.16
      3635648.61     10197602.55      3635049.71     10199086.78
#Sta/Elev= 30
    1195  287.09  1318.2  277.28  1694.4  235.68  1909.3  217.37  2043.7  215.26
  2335.7  215.43  2394.3  224.77    2449   215.1  2595.4  212.25    2864  210.12
  2997.9  209.01  3269.9  207.03  3371.3  205.43  3593.9   205.3  4482.3  208.82
  4781.5  209.66  4852.9   200.9    4914  206.26    4980  204.76  5002.8  193.92
  5005.6  193.42  5008.8  193.92  5046.6  208.64  5094.8  208.06  5608.3  207.05
  6338.1  207.79  6635.2  207.52  6739.5  213.41  6940.7  226.89  7170.8  233.21
#Mann= 20 ,-1 , 0
    1195     .08       0  1318.2     .05       0  1694.4     .08       0
  1909.3     .12       0  2043.7     .05       0    2449     .12       0
  2595.4     .16       0    2864     .05       0  2997.9     .16       0
  3269.9     .12       0  3371.3     .16       0  3593.9     .16       0
  4482.3     .12       0  5002.8     .07       0  5008.8     .12       0
  5094.8     .16       0  5608.3     .05       0  6338.1     .16       0
  6635.2      .1       0  6739.5     .05       0
Bank Sta=4914,5046.6
XS Rating Curve= 0 ,0
Exp/Cntr=0.3,0.1

Type RM Length L Ch R = 1 ,41732   ,1840,1840,1840
XS GIS Cut Line= 2
     3637271.098    10194258.431     3633529.778    10197574.403
#Sta/Elev= 30
       0  317.17  309.72  311.84   559.5  291.71  679.39  271.29  729.34  265.96
  859.23  238.38 1009.09  225.01 1079.03  213.57 1338.79  213.77 1388.75  224.32
 1458.68  208.02 1538.61  203.65  2657.6  205.99 2797.48  203.58 2837.44  205.97
 3376.96  206.91 3416.92  199.17 3456.88  206.03 3586.77  206.96 3626.73  200.18
 3646.71  192.44 3666.69  191.71 3706.66  204.21 3736.63  207.69 3976.41  205.68
 4455.98  213.42 4585.87  211.18 4705.76  213.05  4885.6  227.47 5045.45  225.21
#Mann= 3 , 0 , 0
       0     .05       0 3586.77     .07       0 3736.63     .05       0
Bank Sta=3586.77,3736.63
XS Rating Curve= 0 ,0
Exp/Cntr=0.3,0.1

Type RM Length L Ch R = 1 ,39874   ,2622,2622,2622
XS GIS Cut Line= 3
     3636823.206    10194146.698     3633527.145    10195575.409
     3633314.092    10197455.292
#Sta/Elev= 30
       0  308.14  209.59  299.21  389.24  287.25  718.59  249.39  848.33   230.9
  978.08  222.81 1047.94  213.27 1297.45  214.15 1337.37  223.15 1357.33  224.34
 1437.18   206.6 1536.98  204.25 2115.84  203.57 2225.63  199.45 2265.55  204.23
 3173.76   200.8  3203.7  208.34 3213.69  208.16 3263.59  203.71 3293.53   190.2
 3303.51  190.03 3333.45  204.39 3353.41  205.54 3862.46  204.26  3952.3  200.02
 4151.94  204.78 4581.17  203.05 5050.33  214.66 5200.06  223.42 5409.69  225.96
#Mann= 3 ,-1 , 0
       0     .05       0  3203.7     .07       0 3353.41     .05       0
Bank Sta=3213.69,3353.41
XS Rating Curve= 0 ,0
Exp/Cntr=0.3,0.1

Type RM Length L Ch R = 1 ,37270   ,508,508,508
XS GIS Cut Line= 2
     3633827.926    10190537.323     3633176.234    10197367.564
#Sta/Elev= 30
       0  268.23  829.49  237.76 1099.32  242.95 1738.93  230.92 2138.69  202.44
 2218.64  202.33  2278.6  209.16 2388.53  200.04 2588.41  203.69 2668.36  198.95
 2698.34  202.99 2818.27  204.25 2888.23  194.58 2948.19  198.33 2968.18  189.98
 2988.16  188.59 3028.14  195.04 3128.08  195.86 3188.04  202.56 4117.47  204.31
 4197.42  200.54 4247.39  204.13 4657.14  202.38 4807.05  208.13 4867.01  203.07
 5876.39  203.34 5916.37  214.33 6046.29  218.58 6266.15  217.52  6835.8  229.92
#Mann= 4 ,-1 , 0
       0     .05       0 2818.27     .07       0 3188.04     .12       0
 4807.05     .05       0
Bank Sta=2818.27,3188.04
XS Rating Curve= 0 ,0
Exp/Cntr=0.3,0.1

Type RM Length L Ch R = 1 ,36762   ,1317,1317,1317
XS GIS Cut Line= 2
     3633339.157    10190612.518     3632925.583    10197129.445
#Sta/Elev= 30
       0  265.32  539.42  219.76  619.34  217.46  709.24  224.27  759.19  218.45
 1238.67  205.58 1448.45  204.91 1518.37  210.61 1598.29  200.71 2737.07  202.71
 2836.96  188.19 2866.93  194.72 3016.77  194.45 3066.71  202.24 3116.66  198.15
 3935.78  200.93 4095.61  207.52 4265.43  198.24 4355.33   203.3 5084.55  200.46
 5114.52  205.23  5504.1  213.41 5613.99  210.44  5693.9  221.51 5793.79  224.81
 5853.73  220.57 5913.66  227.42 6203.35  234.37 6393.15  245.66 6513.02  245.19
#Mann= 4 ,-1 , 0
       0     .05       0 2737.07     .07       0 3066.71     .12       0
 5114.52     .05       0
Bank Sta=2737.07,3066.71
XS Rating Curve= 0 ,0
Exp/Cntr=0.3,0.1

Type RM Length L Ch R = 1 ,35445   ,769,769,769
XS GIS Cut Line= 3
     3633289.027    10190599.986     3631998.174    10194033.905
     3630983.037    10195550.344
#Sta/Elev= 30
       0  268.57   49.89  267.93  628.55  215.39  708.37  220.41  838.07  213.15
 1047.59   213.7 1107.45  202.58 1147.36  200.93 1825.79  197.99 2005.38  201.33
 2055.26  187.08 2105.15  201.56 2274.76   198.4 2514.21  200.74 2544.14  197.29
  2993.1  201.07 3112.83  196.87 3142.76  200.83 3641.61  201.04  3701.5   196.9
 3771.42  200.84 4210.95  200.72 4290.86  215.39 4340.81  208.52 4680.44  208.86
 4870.24  220.21  5000.1  213.25 5249.83  220.82 5349.72  231.93 5479.58  231.84
#Mann= 4 ,-1 , 0
       0     .05       0 2005.38     .07       0 2105.15     .12       0
 4290.86     .05       0
Bank Sta=2005.38,2105.15
XS Rating Curve= 0 ,0
Exp/Cntr=0.3,0.1

Type RM Length L Ch R = 1 ,34676   ,961,961,961
BEGIN DESCRIPTION:
GIBBONS CREEK 23.0
END DESCRIPTION:
XS GIS Cut Line= 3
      3633174.64     10190454.13      3632145.24     10191545.99
      3630942.11     10195091.62
#Sta/Elev= 30
  2842.9   278.6  2956.1  281.33  3033.8  275.95  3404.3  232.75  3543.2  213.19
  3586.7  217.84  3663.7  214.26  3691.6  206.81    3739  202.22  3958.6  201.88
  4550.1  198.11  4828.5  199.15  4861.9   199.1  4951.4  200.92  4986.8  186.92
  4989.6  186.42  4992.8  186.92  5046.4   200.6  5206.1  198.25  5617.9  199.26
  5722.3  195.82  6246.3  198.14  6343.1  198.51  6824.1  199.06  6978.3  199.99
  7046.4  216.42  7109.2  208.43  7718.1  208.33  8003.2  213.19  8087.7  219.65
#Mann= 15 ,-1 , 0
  2842.9     .05       0  3404.3      .1       0  3586.7     .05       0
    3739     .12       0  3958.6     .16       0  4550.1     .12       0
  4828.5     .16       0  4861.9     .12       0  4986.8     .07       0
  4992.8     .12       0  5206.1     .16       0  5617.9     .12       0
  6246.3     .16       0  6343.1     .12       0  6824.1     .05       0
Bank Sta=4951.4,5046.4
XS Rating Curve= 0 ,0
Exp/Cntr=0.3,0.1

Type RM Length L Ch R = 1 ,33715   ,1506,1506,1506
BEGIN DESCRIPTION:
GIBBONS CREEK 22.0
END DESCRIPTION:
XS GIS Cut Line= 3
      3632842.08     10190191.67       3629893.4     10192928.07
      3627380.34     10193865.59
#Sta/Elev= 30
  2619.9  297.82    2818  283.65  3243.9  223.72  3312.9  213.99  3382.6  213.76
  3521.2  200.33  3592.3  198.72  4075.7  197.29  4214.3  198.06    4353  197.58
  4570.6  196.56  4947.9  199.51  4994.3   186.3    4997   185.8  5000.3   186.3
  5025.6  199.09  5184.8  197.03  5323.4  197.31  5754.2  198.35  6157.8  196.89
  6207.8   206.5  6440.7  228.91  6878.9  214.69  7302.4  215.35  7409.4  215.46
  7683.9  224.08    8044  242.57  8466.7  214.86  8596.3   219.4  9324.9  259.32
#Mann= 20 ,-1 , 0
  2619.9     .05       0  3243.9     .08       0  3312.9      .1       0
  3382.6     .05       0  3521.2     .16       0  3592.3     .05       0
  4075.7     .12       0  4214.3     .12       0    4353     .12       0
  4570.6     .12       0  4994.3     .07       0  5000.3     .12       0
  5184.8     .16       0  5323.4     .16       0  5754.2     .12       0
  6207.8     .05       0  7302.4     .08       0  7409.4     .05       0
  7683.9     .16       0  8596.3     .05       0
#XS Ineff= 1 ,-1
 6445.45 9568.18  229.26
Permanent Ineff=
       F
Bank Sta=4947.9,5025.6
XS Rating Curve= 0 ,0
Exp/Cntr=0.3,0.1

Type RM Length L Ch R = 1 ,32209   ,2277,2277,2277
BEGIN DESCRIPTION:
GIBBONS CREEK 21.0
END DESCRIPTION:
XS GIS Cut Line= 3
      3632106.94     10189555.67      3629502.78     10191625.99
      3627198.07     10193084.34
#Sta/Elev= 30
  2613.9   285.1  2866.8  276.28    2908   274.2  3054.3  253.47    3263   225.1
  3428.6  211.79  3454.2  209.66  3489.2  198.54  3567.7  194.52  4758.3  195.36
  4882.4  196.78  4970.7  197.36  5003.2  185.86    5006  185.36  5009.2  185.86
  5055.9  198.59  5198.4  198.41  5219.2  191.19  5446.5  196.79  5494.3  196.12
  5641.1  196.47  6024.3   195.9  6213.8  197.59  6263.8  197.29  6353.6  197.71
  6466.9  197.56  6582.2  220.18  8228.6   214.9  8249.3  214.93  8668.1  231.17
#Mann= 20 ,-1 , 0
  2613.9     .05       0  2866.8     .08       0    2908     .05       0
  3054.3      .1       0    3263     .05       0  3428.6      .1       0
  3454.2     .16       0  4758.3     .12       0  4882.4     .12       0
  5003.2     .07       0  5009.2     .12       0  5446.5     .16       0
  5494.3     .12       0  5641.1     .16       0  6024.3     .12       0
  6213.8     .16       0  6263.8     .12       0  6353.6     .05       0
  8228.6     .08       0  8249.3     .05       0
#XS Ineff= 1 ,-1
 6581.82 8538.64     221
Permanent Ineff=
       F
Bank Sta=4970.7,5055.9
XS Rating Curve= 0 ,0
Exp/Cntr=0.3,0.1

Type RM Length L Ch R = 1 ,29932   ,1634,1634,1634
BEGIN DESCRIPTION:
GIBBONS CREEK 20.0
END DESCRIPTION:
XS GIS Cut Line= 3
      3631182.48     10188487.96      3628083.51     10190206.72
      3626651.24     10191886.37
#Sta/Elev= 30
  2106.3  263.43  2139.8  264.37  2160.6  265.69  2330.1  270.89  2852.9  249.47
  2968.2  237.84  3219.3  206.31  3294.8  212.18    3344  202.41  3449.2  200.14
  3822.7  198.58  4118.9  190.11  4954.3  196.44  4989.1  186.19  4991.8  185.69
  4995.1  186.19  5035.6  195.51  5388.6  188.73  6254.1  191.41    6323  192.72
  6706.6  197.93  6831.6  203.77  6886.7  205.61  6956.6  206.73  7046.2  207.22
  7331.6  212.28  7365.1  212.31  7456.5  214.99  7831.5  223.66  7857.4  223.74
#Mann= 20 ,-1 , 0
  2106.3     .05       0  2139.8      .1       0  2160.6     .05       0
  2852.9     .08       0  2968.2     .05       0  3449.2     .16       0
  3822.7     .12       0  4989.1     .07       0  4995.1     .12       0
  6254.1     .05       0    6323     .12       0  6706.6      .1       0
  6831.6     .05       0  6886.7      .1       0  6956.6     .05       0
  7046.2     .16       0  7331.6      .1       0  7365.1     .05       0
  7456.5     .16       0  7831.5     .05       0
Bank Sta=4954.3,5035.6
XS Rating Curve= 0 ,0
Exp/Cntr=0.3,0.1

Type RM Length L Ch R = 1 ,28298   ,1615,1615,1615
BEGIN DESCRIPTION:
GIBBONS CREEK 20.2
END DESCRIPTION:
XS GIS Cut Line= 3
      3629945.49     10187537.45      3626574.28     10189575.46
       3625011.4     10191247.51
#Sta/Elev= 30
  2481.1  269.13  2625.3  264.85  2723.1  252.12  2888.9  228.32  3079.2   206.2
  3410.7  211.96  3490.3  193.25  3668.1   192.6  3965.1  193.58  4083.3  192.83
  4121.3  193.11  4876.5  193.27  4970.6  193.61  5010.3  185.02  5013.1  184.52
  5016.3  185.02  5034.7  193.29  5158.2  191.99  5198.7  190.69  5647.7  195.11
  5990.6  186.93  6117.9  193.17    6908  191.78  7050.7  191.64  7812.9  198.12
  7905.2  210.31  8188.1   220.1  8301.4  216.35  8602.3  236.44  8709.2  238.35
#Mann= 17 ,-1 , 0
  2481.1      .1       0  2723.1     .05       0  2888.9      .1       0
  3079.2     .05       0  3668.1     .16       0  3965.1      .1       0
  4083.3     .12       0  4121.3      .1       0  4876.5     .12       0
  5010.3     .07       0  5016.3     .12       0  5158.2     .16       0
  5198.7     .12       0  6117.9      .1       0    6908     .05       0
  7050.7      .1       0  8602.3     .16       0
Bank Sta=4970.6,5034.7
XS Rating Curve= 0 ,0
Exp/Cntr=0.3,0.1

Type RM Length L Ch R = 1 ,26683   ,3625,3625,3625
BEGIN DESCRIPTION:
GIBBONS CREEK 20.1
END DESCRIPTION:
XS GIS Cut Line= 4
      3629711.11      10186508.8      3627484.55     10187498.38
      3626234.55     10188084.32      3623578.28     10190584.34
#Sta/Elev= 30
  2053.4  238.19  2252.7  243.19  2389.4     244  2468.9  233.93  2676.1  205.87
  3356.5  205.46  3387.4  211.82    3464  194.14  3604.5  190.38  4273.7  190.51
  4411.4  190.86  4840.3  192.49    4954  191.81  4996.7  184.17  4999.4  183.67
  5002.7  184.17    5028  191.64  5331.2  191.55  5489.5  190.75  5518.4  184.71
    6030  189.93  6126.7  189.08  6554.7  192.23  8095.3  194.08  8288.8  196.43
  8391.8  197.68    8711  206.65  8870.2  217.04  9414.7  236.83  9518.2  243.42
#Mann= 20 ,-1 , 0
  2053.4     .05       0  2252.7     .05       0  2468.9     .05       0
  3604.5      .1       0  4273.7     .12       0  4411.4      .1       0
  4840.3     .12       0  4996.7     .07       0  5002.7     .12       0
  5331.2     .16       0  5489.5     .12       0    6030     .16       0
  6126.7     .12       0  6554.7      .1       0  8095.3     .16       0
  8288.8     .16       0  8391.8      .1       0    8711     .16       0
  8870.2      .1       0  9414.7     .05       0
Bank Sta=4954,5028
XS Rating Curve= 0 ,0
Exp/Cntr=0.3,0.1

Type RM Length L Ch R = 1 ,23058   ,2529,2529,2529
BEGIN DESCRIPTION:
GIBBONS CREEK 19.0
END DESCRIPTION:
XS GIS Cut Line= 5
      3629294.42     10185011.42      3627875.17      10185818.7
      3626208.51     10186066.09      3624406.23     10186358.29
      3622862.19     10187290.03
#Sta/Elev= 30
  1219.6   245.9  1514.5  245.02  1750.9  267.68  1918.1  262.99    2493  203.93
  2618.6  194.45  2845.2  188.58  3211.1   188.7  3445.2  189.02  3645.9  189.76
  3761.6  189.69  4135.6  189.46  4263.2  189.87  4448.9  190.96  4523.1  191.18
  4969.3   188.9  4996.7  181.29  4999.4  180.79  5002.7  181.29  5009.1  183.88
  5030.1  190.47  5405.7  192.46  5516.3   188.7  5587.2  205.26  5857.5  199.42
  6092.5  204.13  6399.2  216.34  6551.2  212.37  6858.5  234.88  8166.5  243.04
#Mann= 20 ,-1 , 0
  1219.6     .05       0    2493     .12       0  2618.6     .07       0
  2845.2     .16       0  3211.1      .1       0  3445.2      .1       0
  3645.9     .12       0  3761.6      .1       0  4135.6     .12       0
  4263.2      .1       0  4448.9     .16       0  4523.1     .12       0
  4996.7     .07       0  5002.7     .07       0  5009.1     .12       0
  5405.7     .05       0  5857.5     .16       0  6092.5     .05       0
  6399.2     .16       0  6858.5     .05       0
#XS Ineff= 1 ,-1
 5586.36 6286.36  205.66
Permanent Ineff=
       F
Bank Sta=4969.3,5030.1
XS Rating Curve= 0 ,0
Exp/Cntr=0.3,0.1

Type RM Length L Ch R = 1 ,20529   ,1481,1481,1481
BEGIN DESCRIPTION:
GIBBONS CREEK 18.0
END DESCRIPTION:
XS GIS Cut Line= 3
      3628838.68     10184620.78      3625509.81     10184822.37
      3623369.98     10185284.84
#Sta/Elev= 30
  2101.7  298.29  2434.9  283.43  2619.6  271.22  2849.6  258.53  3009.9  259.61
  3230.3  230.88  3320.5  238.47  3420.7   214.8  3536.5  200.26  3651.1  185.15
    3773  188.12    4797  187.01  4893.4  184.53  4953.5  189.99  4990.6  179.93
  4993.3  179.43  4996.6  179.93  5053.7  188.01  5113.8  190.37  5163.9  207.33
  5216.3  216.07  5436.7  222.96  5595.9  207.52  5700.3  209.42  5751.5  199.48
  6099.3  199.25    6545  234.18  6948.5  237.95  7614.3  233.69  7625.9  233.72
#Mann= 10 ,-1 , 0
  2101.7     .16       0  2434.9      .1       0  2619.6     .16       0
  3536.5     .12       0    3773      .1       0    4797     .12       0
  4990.6     .07       0  4996.6     .12       0  5216.3     .05       0
  7614.3     .08       0
#XS Ineff= 1 ,-1
 5432.95 6588.64  223.08
Permanent Ineff=
       F
Bank Sta=4953.5,5053.7
XS Rating Curve= 0 ,0
Exp/Cntr=0.3,0.1

Type RM Length L Ch R = 1 ,19048   ,1205,1205,1205
BEGIN DESCRIPTION:
GIBBONS CREEK 17.0
END DESCRIPTION:
XS GIS Cut Line= 3
      3628200.66     10183409.84      3626169.44      10183448.9
       3623956.5     10184529.34
#Sta/Elev= 30
  2630.6  255.69  2779.2  255.53  3079.2  218.95  3346.7  197.26  3919.4  189.43
  4275.1  189.68  4472.6  187.03  4566.9  186.95  4662.2  187.61  4728.5  183.49
  4790.5  187.55  4953.7  189.42  5001.3  179.48  5004.1  178.98  5007.3  179.48
  5049.4  187.18  5297.2  186.26  5326.9  190.87  5357.9  190.55  5516.1  191.22
  5582.9  205.28  5612.5   199.8  5858.7  199.48  6210.1  201.29  6389.5  204.37
  6450.9  208.92  6592.2  230.91  6727.3   242.5  6817.4  243.14  7124.8  233.25
#Mann= 10 ,-1 , 0
  2630.6     .16       0  3346.7     .12       0  4275.1     .16       0
  4472.6      .1       0  4566.9     .12       0  5001.3     .07       0
  5007.3     .12       0  5357.9     .05       0  5858.7     .16       0
  6210.1     .05       0
#XS Ineff= 1 ,-1
 5586.36 6564.77  205.56
Permanent Ineff=
       F
Bank Sta=4953.7,5049.4
XS Rating Curve= 0 ,0
Exp/Cntr=0.3,0.1

Type RM Length L Ch R = 1 ,17843   ,1667,1667,1667
BEGIN DESCRIPTION:
GIBBONS CREEK 15.0
END DESCRIPTION:
XS GIS Cut Line= 3
      3627237.16     10180349.94      3625010.59     10183227.55
      3624021.03     10183722.33
#Sta/Elev= 30
  1847.8  238.67  1898.2   237.7  2030.5  243.48  2088.4  235.94  2258.6  242.27
  2642.2  233.38  2843.6  230.22  3127.9  237.79  3285.5  220.04  3414.1   223.6
  3727.3  206.53  4346.7  189.84  4439.5  188.23  4792.1  188.98    4947  189.61
  4993.8  178.93  4996.6  178.43  4999.8  178.93  5009.4  183.08  5017.7  186.73
  5120.5  185.82  5251.1   183.9  5378.2  189.83  5627.9  193.33  5800.2  214.95
  5844.9  211.11  5884.1  219.75  6032.9  221.27  6145.5  221.27  6592.6  226.82
#Mann= 15 ,-1 , 0
  1847.8     .05       0  1898.2      .1       0  2642.2     .05       0
  4346.7      .1       0  4439.5     .05       0  4792.1     .12       0
  4993.8     .07       0  4999.8     .12       0  5009.4     .05       0
  5120.5     .12       0  5251.1     .05       0  5378.2     .12       0
  5627.9     .05       0  6032.9     .08       0  6145.5     .05       0
Bank Sta=4947,5017.7
XS Rating Curve= 0 ,0
Exp/Cntr=0.3,0.1

Type RM Length L Ch R = 1 ,16176   ,1196,1196,1196
BEGIN DESCRIPTION:
GIBBONS CREEK 13.0
END DESCRIPTION:
XS GIS Cut Line= 3
      3626260.59      10180636.4      3624554.86      10182198.9
      3623591.31     10183084.33
#Sta/Elev= 30
  3197.9  263.03  3547.6  269.21  3603.7  264.09  3731.4  260.01  4129.3  259.35
  4184.6  256.41  4205.6  248.45  4219.7  248.62  4226.5  244.24  4233.9  244.73
  4283.3  230.51    4340  223.46  4722.3  194.87  4793.6  192.83  4913.5  185.01
  4948.6  180.12  4963.8  181.23  5002.3  179.18  5005.1  178.68  5008.3  179.18
  5033.7  185.53  5191.9  187.95  5231.7   190.2  6045.6  187.42  6300.8  195.02
  6364.3  207.28  6498.7  205.47  6661.6  217.38  6710.8   222.2  6819.7  222.62
#Mann= 8 ,-1 , 0
  3197.9     .05       0  4129.3     .16       0  4793.6     .05       0
  4963.8     .12       0  5002.3     .07       0  5008.3     .12       0
  5191.9     .05       0  6661.6     .08       0
Bank Sta=4913.5,5033.7
XS Rating Curve= 0 ,0
Exp/Cntr=0.3,0.1

Type RM Length L Ch R = 1 ,14980   ,910,910,910
BEGIN DESCRIPTION:
GIBBONS CREEK 11.0
END DESCRIPTION:
XS GIS Cut Line= 3
      3625518.36     10180662.46       3624268.4     10181053.07
      3622497.56     10182211.93
#Sta/Elev= 30
  3344.2  245.94  3492.3  238.53  3568.5  241.88  3811.7  251.32  3930.2  242.08
  4073.7  220.19  4144.2  214.53  4395.4  194.38  4595.5   186.3  4678.9  185.65
  4829.6  189.84  4878.5  186.94    4896  185.29  4968.4  187.86  5007.6  179.27
  5010.3  178.77  5013.6  179.27    5014  179.29  5031.8  179.69  5061.9   189.9
  5143.3  188.83  5281.8  187.07  6080.4  187.92  6242.8   193.8  6433.9  199.97
  6491.1  212.76  6527.3  208.91  6557.5  213.67  6608.8  213.75  6770.1  205.38
#Mann= 11 ,-1 , 0
  3344.2     .05       0  3568.5     .16       0  4144.2     .05       0
  4878.5     .12       0  5007.6     .07       0  5013.6     .12       0
    5014     .05       0  5143.3     .08       0  5281.8     .05       0
  6080.4     .12       0  6242.8     .05       0
Bank Sta=4968.4,5061.9
XS Rating Curve= 0 ,0
Exp/Cntr=0.3,0.1

Type RM Length L Ch R = 1 ,14070   ,1214,1214,1214
BEGIN DESCRIPTION:
GIBBONS CREEK 10.0
END DESCRIPTION:
XS GIS Cut Line= 3
      3626888.64      10179453.5      3624572.45     10179974.22
      3622081.79     10181374.08
#Sta/Elev= 30
  1850.2  233.09  2061.9  236.69  2123.4  230.76  2186.8  238.46  2230.1  233.55
  2297.6  240.78  2505.3  244.67  2769.1  233.46  2808.3  237.88  3012.4  232.08
  3313.3  214.39  3503.9  204.31  4189.2  188.78  4800.8  189.81  4855.5  190.15
  4982.9   178.7  4985.6   178.2  4988.9   178.7  4994.6  180.36  5073.5  190.08
  5258.5  188.37  5393.4  188.22  6138.2  185.01  6183.5  185.02  6279.4  184.78
  6449.6  190.75  6610.6  209.77    6645  207.52  6800.3   220.3  7081.3  218.87
#Mann= 14 ,-1 , 0
  1850.2     .05       0  2808.3     .08       0  3012.4     .16       0
  3313.3     .05       0  4800.8     .12       0  4982.9     .03       0
  4988.9     .12       0  4994.6     .05       0  5258.5     .08       0
  5393.4     .05       0  6138.2     .12       0  6183.5     .05       0
  6279.4     .12       0  6449.6     .05       0
Bank Sta=4855.5,5073.5
XS Rating Curve= 0 ,0
Exp/Cntr=0.3,0.1

Type RM Length L Ch R = 1 ,12856   ,2597,2597,2597
BEGIN DESCRIPTION:
GIBBONS CREEK 8.0
END DESCRIPTION:
XS GIS Cut Line= 3
      3626183.37     10177305.07      3624458.13     10178661.39
      3621702.03     10181243.88
#Sta/Elev= 30
  2096.8  222.56  2215.9  222.96  2443.7  212.13  2515.9  213.41  2700.3  197.76
  3021.1  191.41    3135  193.01  3932.1  183.83  4444.4  184.65    4916  189.57
  4946.5  189.65  4974.9  184.71  4982.2  178.85  5007.5  178.59  5010.3  178.09
  5013.5  178.59  5056.4  185.97  5109.2  184.53  5151.7  189.65  5164.7  189.92
  6941.9  185.26  7118.7   200.5  7153.9  208.45  7196.4  205.16  7238.9  211.07
  7373.2  218.23  7458.2  220.57  7550.1  217.97  7868.5  225.83  8068.3  219.19
#Mann= 6 ,-1 , 0
  2096.8     .05       0    4916     .16       0  5007.5     .07       0
  5013.5     .16       0  5056.4     .12       0  5164.7     .05       0
Bank Sta=4946.5,5151.7
XS Rating Curve= 0 ,0
Exp/Cntr=0.3,0.1

Type RM Length L Ch R = 1 ,10259   ,2080,2080,2080
BEGIN DESCRIPTION:
GIBBONS CREEK 7.0
END DESCRIPTION:
XS GIS Cut Line= 3
      3624021.01     10175805.67      3621859.55     10178865.57
      3621364.75     10180584.35
#Sta/Elev= 30
  1551.7  219.61  1712.3  213.33  1900.4   206.6  1927.4  202.95  1988.8  207.61
  2158.9  206.48  2531.5  188.76  2681.5  183.46  2947.8  183.23  3885.7   184.6
  3936.6  184.74  4287.8  185.07  4406.7  185.18  4916.9  188.06  4920.4   188.1
    4977  183.88  4999.4  177.55  5036.1  179.99  5095.9   177.5  5098.6     177
  5101.9   177.5  5178.9  187.14  5335.6  183.18  5386.6   185.2    5995  192.06
    6319  200.64  6448.2  209.51  6549.3  202.15  6698.8  202.63  7086.6  213.63
#Mann= 16 ,-1 , 0
  1551.7     .05       0  1712.3     .16       0  1988.8     .05       0
  2531.5     .16       0  2681.5     .12       0  2947.8     .05       0
  3885.7     .16       0  3936.6     .05       0  4287.8      .1       0
  4406.7     .16       0  4916.9     .12       0  5095.9     .07       0
  5101.9     .12       0  5386.6     .05       0  6448.2     .08       0
  6549.3     .05       0
Bank Sta=4920.4,5178.9
XS Rating Curve= 0 ,0
Exp/Cntr=0.3,0.1

Type RM Length L Ch R = 1 ,8179    ,1114,1114,1114
BEGIN DESCRIPTION:
GIBBONS CREEK 6.0
END DESCRIPTION:
XS GIS Cut Line= 3
      3622679.87     10175441.06      3621742.36     10177368.17
      3620166.99      10180440.8
#Sta/Elev= 30
  3218.7  213.82  3947.9   190.3    3997  188.48  4211.3  182.45  4797.6  187.11
  4843.4  185.98  4973.4  177.18  4976.1  176.68  4979.4  177.18  4989.6  177.32
  5034.2  187.53  5631.5  184.27  6072.2  187.44  6182.3   180.1  6226.7   187.6
  6397.2   186.1  6505.3  184.98  6687.7  185.09  6830.1  185.58  6912.2  185.35
  7120.7   186.3  7148.6  186.38  7258.7  186.96  7386.3  199.24  7480.7  191.38
  7696.3  193.76  7868.1  195.34  7920.8   195.7  8234.2  199.02  8814.7  212.59
#Mann= 20 ,-1 , 0
  3218.7     .05       0  3947.9     .12       0    3997     .05       0
  4843.4     .12       0  4973.4     .07       0  4979.4     .12       0
  4989.6     .16       0  5631.5     .05       0  6072.2     .12       0
  6397.2     .05       0  6505.3     .16       0  6687.7     .05       0
  6830.1     .08       0  6912.2     .05       0  7120.7     .16       0
  7148.6     .05       0  7696.3      .1       0  7868.1     .05       0
  7920.8      .1       0  8234.2     .05       0
#XS Ineff= 1 ,-1
 7384.09  8437.5  199.18
Permanent Ineff=
       F
Bank Sta=4797.6,5034.2
XS Rating Curve= 0 ,0
Exp/Cntr=0.3,0.1
