HEC-RAS study NAVASOTA RIVER.prj: NAVASOTA RIVER Base Level Engineering

--- NAVASOTA RIVER.g01 (geometry) --- (continued)

Type RM Length L Ch R = 1 ,425247  ,1758,1758,1758
BEGIN DESCRIPTION:
NAVASOTA RIVER 359
END DESCRIPTION:
XS GIS Cut Line= 3
      3593949.96     10331635.47      3590300.98      10329561.1
      3587197.34      10328985.3
#Sta/Elev= 30
   802.6  296.08   859.3  293.41  1048.7  284.28  1159.8  279.21  1197.8  277.44
    1271  273.76  1444.8     267  1961.2  257.95  2493.5  251.21  2691.9  251.93
  4124.5  244.99    4926  252.42  4990.6  236.99  5059.9  251.95  5794.6  254.92
  5953.1  243.35  6073.2   254.8  6691.1   258.1  6776.2  241.79  6834.1   254.3
  7043.1   243.9  7073.7  254.59  7137.6  252.22  7205.9  259.36  7291.8  251.61
    7330  244.77  7368.6  254.76  7566.9  255.42  7744.9  275.01  8156.6   275.7
#Mann= 17 ,-1 , 0
   802.6     .16       0   859.3     .05       0  1048.7     .16       0
  1159.8     .12       0  1197.8     .16       0    1271     .12       0
  1444.8     .05       0  1961.2     .12       0  2493.5     .05       0
  2691.9     .12       0    4926     .07       0  5059.9     .12       0
  6073.2     .05       0  6691.1     .16       0  7137.6     .05       0
  7291.8     .12       0  7566.9     .16       0
#XS Ineff= 2 , 0
       0                  6514.3       0  261.68
Permanent Ineff=
       F       F
Bank Sta=4926,5059.9
XS Rating Curve= 0 ,0
Exp/Cntr=0.3,0.1

Type RM Length L Ch R = 1 ,423489  ,1408,1408,1408
BEGIN DESCRIPTION:
NAVASOTA RIVER 360
END DESCRIPTION:
XS GIS Cut Line= 3
      3595922.23     10330809.11      3591629.14     10328818.12
      3587498.97     10328027.83
#Sta/Elev= 30
   267.7  295.47   718.2  276.08   873.3  271.38  1333.7   265.3    1491  262.07
  1676.9  257.91  2251.9  251.64  2923.1  249.87  3032.2  249.92  3200.5  248.45
  3299.2  251.13  3315.8  246.95  3504.6  244.93  3693.4  251.81  4492.6  251.57
  4607.5  250.48    4758  251.17  4957.1  251.67  4974.5   239.6  5009.8  236.16
  5037.7  238.81  5068.3  251.23  5868.6  252.26  6057.9  253.33  6284.7   252.5
  7597.4  253.28  8516.1  254.58  8631.8  255.12  8834.6  275.72  9205.1  274.25
#Mann= 20 ,-1 , 0
   267.7     .16       0   718.2     .05       0   873.3     .16       0
  1333.7     .12       0    1491     .16       0  1676.9     .05       0
  2251.9     .12       0  2923.1     .05       0  3032.2     .07       0
  3200.5     .12       0  4492.6     .07       0  4607.5     .12       0
    4758     .12       0  4957.1     .07       0  5068.3     .12       0
  5868.6     .12       0  6057.9     .05       0  6284.7     .05       0
  7597.4     .05       0  8516.1     .16       0
Bank Sta=4957.1,5068.3
XS Rating Curve= 0 ,0
Exp/Cntr=0.3,0.1

Type RM Length L Ch R = 1 ,422081  ,4921,4921,4921
BEGIN DESCRIPTION:
NAVASOTA RIVER 361
END DESCRIPTION:
XS GIS Cut Line= 3
      3598577.35     10328309.96      3591762.06     10327426.62
      3586276.67     10326958.87
#Sta/Elev= 30
 -1872.3  346.37 -1864.5   345.4 -1574.6  323.05 -1225.4  298.15  -515.8  289.93
    -369  270.23  -136.3  261.43  2687.1   248.2  3002.2  248.35  3365.2  250.48
  3406.7  244.95  3470.4  250.57  3656.4  248.96    4647  251.99  4690.5  246.65
  4939.5  253.15  4999.7  236.06  5030.1  238.38  5070.2  252.86  5098.7  252.74
  5253.1  251.75    6615  251.35  8382.2  250.94  8723.4   267.5  8990.8  265.92
  9000.6   266.2  9089.6  265.94  9951.7  266.76 10248.9  264.78 10505.3  276.77
#Mann= 17 ,-1 , 0
 -1872.3     .05       0 -1864.5     .16       0 -1574.6     .05       0
  2687.1     .12       0  3002.2     .05       0  3365.2     .12       0
  3470.4     .05       0  3656.4     .12       0  4939.5     .07       0
  5070.2     .12       0  5098.7     .16       0  5253.1     .12       0
    6615     .05       0  8990.8      .1       0  9000.6     .05       0
  9089.6     .16       0  9951.7     .05       0
#XS Ineff= 2 , 0
       0  -527.4  290.31               0
Permanent Ineff=
       F       F
Bank Sta=4939.5,5070.2
XS Rating Curve= 0 ,0
Exp/Cntr=0.3,0.1

Type RM Length L Ch R = 1 ,417160  ,3528,3528,3528
BEGIN DESCRIPTION:
NAVASOTA RIVER 362
END DESCRIPTION:
XS GIS Cut Line= 2
      3596984.48     10325355.53      3586255.12     10326787.56
#Sta/Elev= 30
  -853.5  314.39    -451  305.62   -56.6  281.13   168.5  270.49   369.6  257.86
  1237.7  248.99  1316.8  248.18  1556.4   246.1  1983.8  243.21    2569  249.59
  2619.4  242.69  2639.6   249.7  2760.6  250.58    4960  251.36  4990.2  236.29
  5030.3  235.62  5053.3  247.19  5111.3  250.86  5255.2   247.3  5257.8  247.17
  6002.4  250.16  6102.6   250.2  6755.7  251.06  6890.8  250.94  7936.1  250.62
    8259  267.51  8845.3  267.04  9620.9  262.14  9720.2  266.82    9971  278.85
#Mann= 17 ,-1 , 0
  -853.5     .05       0    -451     .16       0   -56.6     .12       0
   168.5     .05       0  1237.7      .1       0  1316.8     .05       0
  1556.4     .12       0    4960     .07       0  5111.3     .12       0
  5255.2     .16       0  5257.8     .12       0  6002.4     .07       0
  6102.6     .05       0  6755.7     .12       0  6890.8     .05       0
  8845.3     .16       0  9720.2     .05       0
#XS Ineff= 2 , 0
       0  3994.5  251.66               0
Permanent Ineff=
       F       F
Bank Sta=4960,5111.3
XS Rating Curve= 0 ,0
Exp/Cntr=0.3,0.1

Type RM Length L Ch R = 1 ,413632  ,3114,3114,3114
BEGIN DESCRIPTION:
NAVASOTA RIVER 363
END DESCRIPTION:
XS GIS Cut Line= 2
      3595407.03     10322792.26      3586042.93     10326069.15
#Sta/Elev= 30
   581.6  296.18  1053.6  290.12    1317  288.28  1483.2  275.65  1720.4  258.91
  2140.9  252.27  2588.5  256.87  2814.1   249.7  3180.4  247.94  3463.9   247.1
  4533.2  247.77  4767.4     248  4955.8  248.92  5004.5  234.93  5036.6   237.3
  5057.7   250.2  5351.1  249.01  5684.6  242.15  5767.1  249.97  6040.7  247.72
  6468.5  248.64  6675.1  250.45  8056.8  249.63  8693.4  248.64  8988.3  265.94
  9598.4  267.12  9932.4  262.85  9984.9  258.85 10285.1  271.31 10502.5  279.34
#Mann= 20 ,-1 , 0
   581.6     .05       0  1053.6      .1       0  1483.2     .12       0
  2140.9     .12       0  2814.1     .07       0  3180.4     .12       0
  3463.9     .12       0  4533.2     .05       0  4767.4     .12       0
  4955.8     .07       0  5057.7     .12       0  5351.1     .12       0
  6040.7     .12       0  6468.5     .07       0  6675.1     .12       0
  8056.8     .12       0  8693.4     .05       0  9598.4     .16       0
  9932.4     .05       0 10285.1     .16       0
Bank Sta=4955.8,5057.7
XS Rating Curve= 0 ,0
Exp/Cntr=0.3,0.1

Type RM Length L Ch R = 1 ,410518  ,3750,3750,3750
BEGIN DESCRIPTION:
NAVASOTA RIVER 391
END DESCRIPTION:
XS GIS Cut Line= 3
      3594085.16     10322046.58      3590432.23     10322593.21
      3586157.98      10324129.9
#Sta/Elev= 30
  1306.4  299.71    1802  270.82  1933.2  260.64  2287.9  255.35  2388.3  256.07
  2507.6  256.16  2655.6  256.04  2890.7  253.33  3292.5  249.37  3392.4  254.21
  3410.8  248.34  3453.1  243.26  4955.1  247.34  4979.9  235.69  5012.9   234.2
  5063.9  247.72  5733.4  246.98  5866.8  240.63  5903.4  246.77  6198.3  246.23
  6734.8  248.94  7978.7  247.96  8088.1  247.91  8194.6  247.73  8459.5  247.29
  8620.5  247.02  8726.9  247.44    8847  247.31  9062.2  268.98  9542.1  272.21
#Mann= 20 ,-1 , 0
  1306.4     .16       0    1802     .05       0  1933.2     .16       0
  2287.9     .07       0  2388.3     .12       0  2507.6     .16       0
  2655.6     .12       0  2890.7     .05       0  3292.5     .07       0
  3410.8     .12       0  4955.1     .07       0  5063.9     .12       0
  6198.3     .05       0  6734.8     .12       0  7978.7     .16       0
  8088.1     .12       0  8194.6     .07       0  8459.5     .12       0
  8620.5     .07       0  8726.9     .05       0
Bank Sta=4955.1,5063.9
XS Rating Curve= 0 ,0
Exp/Cntr=0.3,0.1

Type RM Length L Ch R = 1 ,406768  ,2249,2249,2249
BEGIN DESCRIPTION:
NAVASOTA RIVER 392
END DESCRIPTION:
XS GIS Cut Line= 3
      3594749.43     10321142.35      3589175.72     10321095.82
       3583267.3     10321611.68
#Sta/Elev= 30
  -573.9  298.85  -287.8  295.33  -126.6  293.35   203.4  265.69   322.7   264.2
   873.5  253.78  1901.3  254.56    2562  255.26  2790.1  255.96  3243.6  252.32
  3483.6  241.71  3836.4  246.76  4050.6  246.24  4883.6  247.78  4983.4  233.85
  5043.8   234.9  5063.9  247.14  6161.7  246.97  6755.7  245.96  7029.9   245.4
  7967.1  245.38  8212.9  245.99  8849.1  246.31  9048.1  246.64  9453.8  247.83
 10084.2  247.74 10298.4  252.07 10537.4  275.99 10725.3  298.64 10930.9  298.23
#Mann= 20 ,-1 , 0
  -573.9     .05       0  -287.8     .16       0   322.7     .05       0
  1901.3     .05       0    2562     .12       0  2790.1     .05       0
  3836.4     .12       0  4050.6     .12       0  4883.6     .07       0
  5063.9     .12       0  6161.7     .05       0  6755.7     .12       0
  7029.9     .05       0  7967.1     .12       0  8212.9     .05       0
  8849.1     .12       0  9048.1     .05       0  9453.8     .05       0
 10084.2     .16       0 10537.4     .05       0
Bank Sta=4883.6,5063.9
XS Rating Curve= 0 ,0
Exp/Cntr=0.3,0.1

Type RM Length L Ch R = 1 ,404519  ,2892,2892,2892
BEGIN DESCRIPTION:
NAVASOTA RIVER 393
END DESCRIPTION:
XS GIS Cut Line= 3
      3595177.03     10319719.32      3588324.94     10319226.32
      3582816.57     10318799.23
#Sta/Elev= 30
 -1869.8  297.58 -1725.5  296.42 -1287.4  276.93  -835.8  261.84  -651.7  253.71
     475  252.55  1352.7  252.55  1694.3   244.7  1872.6  247.55  2266.5  248.94
  2766.2   250.1  3480.9  246.13  3669.4  243.77  3970.2  250.63  4180.7  241.87
  4932.7  247.72  4972.5  234.09    5053  235.53  5093.1  247.57  5465.5  245.23
  5786.2   242.5  6249.2  245.05  6560.8  243.16  9230.6  251.68  9392.5  249.11
  9477.3  253.82  9671.9  260.64  9867.4  279.73 10511.4   320.2 10524.9  320.31
#Mann= 20 ,-1 , 0
 -1869.8     .16       0 -1725.5     .05       0 -1287.4     .16       0
  -835.8     .05       0     475     .16       0  1352.7     .12       0
  1872.6     .12       0  2266.5     .12       0  2766.2     .12       0
  3480.9     .12       0  4932.7     .07       0  5093.1     .12       0
  5465.5     .05       0  5786.2     .12       0  6249.2     .05       0
  6560.8     .05       0  9230.6     .16       0  9477.3     .05       0
  9671.9     .16       0 10511.4     .16       0
#XS Ineff= 2 , 0
       0                    9065       0   252.6
Permanent Ineff=
       F       F
Bank Sta=4932.7,5093.1
XS Rating Curve= 0 ,0
Exp/Cntr=0.3,0.1

Type RM Length L Ch R = 1 ,401627  ,2935,2935,2935
BEGIN DESCRIPTION:
NAVASOTA RIVER 394
END DESCRIPTION:
XS GIS Cut Line= 3
      3596055.18     10318908.21      3588566.61     10317045.76
      3582006.41     10316199.97
#Sta/Elev= 30
 -2716.7  296.73 -2244.8  287.06 -1593.5  264.33  -147.7  265.59   184.5  248.93
   268.7  245.29   452.2  244.55  1926.5  244.33  1963.4  244.56  2095.3  244.67
  2263.9  242.72  2962.6   246.6  4325.5  247.51  4942.8  246.32  4973.5  234.37
  5034.8  234.98    5065  246.21  5352.3   245.2  5859.6   248.1  5992.7  240.35
  6918.8  241.69  8669.2  242.65  9471.2  247.61  9521.6  254.37    9562  248.18
 10073.8  249.64 11196.1  275.48 11329.6  295.22 11507.9  341.31 11614.5  338.26
#Mann= 17 ,-1 , 0
 -2716.7     .05       0 -2244.8     .16       0   184.5     .12       0
   268.7     .16       0   452.2     .12       0  1926.5     .16       0
  1963.4     .12       0  2095.3     .16       0  2263.9     .12       0
  2962.6     .16       0  4325.5     .12       0  4942.8     .07       0
    5065     .12       0  5352.3     .05       0  5859.6     .12       0
  6918.8     .05       0 11196.1     .16       0
#XS Ineff= 2 , 0
       0                  9521.6       0  254.37
Permanent Ineff=
       F       F
Bank Sta=4942.8,5065
XS Rating Curve= 0 ,0
Exp/Cntr=0.3,0.1

Type RM Length L Ch R = 1 ,398692  ,2993,2993,2993
BEGIN DESCRIPTION:
NAVASOTA RIVER 395
END DESCRIPTION:
XS GIS Cut Line= 3
       3596415.6     10317501.61      3590561.12     10315813.14
       3586949.8     10314723.22
#Sta/Elev= 30
 -1093.1  296.61  -673.1  286.82  -426.8  272.26  -298.3   266.7   -59.1  255.97
    45.5  261.64   180.3  261.61   264.4  250.81   331.7  260.03   482.1  261.57
   800.4  242.75  1199.6  244.01  1344.3  242.84    2030  242.79  2242.6  242.17
  2724.3  242.76  4957.3  245.69  4996.9  234.23  5056.8  245.64  6325.5  244.24
  6366.9  233.67  6398.7  235.45  6410.6  244.15  6444.7  243.65  6693.7  242.75
  7470.7  240.41  8085.1   243.3  8533.2  282.18  8667.6  294.61  8772.2  299.74
#Mann= 19 ,-1 , 0
 -1093.1     .16       0  -426.8     .05       0  -298.3      .1       0
    45.5     .16       0  1199.6     .12       0  1344.3      .1       0
    2030      .1       0  2242.6     .05       0  2724.3     .12       0
  4957.3     .07       0  5056.8     .12       0  6325.5     .07       0
  6410.6     .12       0  6444.7     .05       0  6693.7     .12       0
  7470.7     .12       0  8085.1     .05       0  8533.2     .16       0
  8667.6     .05       0
#XS Ineff= 2 , 0
       0                  6273.5       0  245.16
Permanent Ineff=
       F       F
Bank Sta=4957.3,5056.8
XS Rating Curve= 0 ,0
Exp/Cntr=0.3,0.1

Type RM Length L Ch R = 1 ,395699  ,2056,2056,2056
BEGIN DESCRIPTION:
NAVASOTA RIVER 192
END DESCRIPTION:
XS GIS Cut Line= 3
      3596892.95     10316400.52       3588299.2     10313557.64
        3586498.     10313535.94
#Sta/Elev= 30
  -836.1   286.7    -656   280.2  -305.9  266.46   163.2  249.18  1531.1  241.66
  1899.1  241.13    2197  242.35    2234  235.07  2265.7  242.37  2376.2  243.12
  2427.6  235.97  2548.3  242.24  2650.7  241.68  4940.7  244.13  4998.9  234.32
  5030.6  242.43  5280.9  242.86    6776  241.97  7198.1  243.06  7377.5  234.13
  7380.3  233.63  7383.5  234.13  7481.5  245.48  7515.8  246.97  8292.8  242.56
  8646.5  253.25  9282.8  285.77  9492.9  281.48  9623.7  291.11   10017  313.97
#Mann= 20 ,-1 , 0
  -836.1     .16       0    -656     .12       0  -305.9     .16       0
   163.2     .12       0  1531.1     .05       0  1899.1     .12       0
  2376.2     .07       0  2427.6     .12       0  2548.3     .07       0
  2650.7     .12       0  4940.7     .07       0  5030.6     .12       0
  5280.9     .12       0    6776     .12       0  7377.5     .07       0
  7383.5     .12       0  7481.5     .07       0  7515.8     .05       0
  8646.5     .16       0  9623.7     .05       0
#XS Ineff= 2 ,-1
  7102.9  7538.5  243.26  7538.5  8552.8  247.95
Permanent Ineff=
       F       F
Bank Sta=4940.7,5030.6
XS Rating Curve= 0 ,0
Exp/Cntr=0.3,0.1

Type RM Length L Ch R = 1 ,393643  ,3421,3421,3421
BEGIN DESCRIPTION:
NAVASOTA RIVER 396
END DESCRIPTION:
XS GIS Cut Line= 3
      3599885.71     10315232.48      3591523.05     10313211.05
      3586726.11     10312800.27
#Sta/Elev= 30
 -3603.5  292.87 -2925.7  239.93 -2496.2  239.17 -2428.5  239.18    1324  240.12
  1505.3   238.9  2099.2  240.11  2405.9  239.91  4949.5  242.22  4990.4  233.09
  5041.1  242.19  5412.4  237.91  6315.7  243.64  6345.9  236.78  6466.3  244.72
  6536.5  235.26  6606.8   234.5    6657  242.56  6818.8  245.99  6908.3  247.49
  7007.1  245.94    7261   244.4  8784.7  249.81  8927.7  256.69  9033.6  264.76
  9186.2  263.58  9359.5  283.76  9457.2  296.19  9527.5  294.14  9814.5  308.23
#Mann= 16 ,-1 , 0
 -3603.5     .16       0 -2925.7     .12       0 -2496.2     .16       0
 -2428.5     .12       0    1324     .07       0  1505.3     .12       0
  2099.2     .07       0  2405.9     .12       0  4949.5     .07       0
  5041.1     .12       0  6818.8     .16       0  6908.3     .05       0
  7007.1     .12       0    7261     .05       0  8927.7     .16       0
  9359.5     .05       0
#XS Ineff= 2 ,-1
  6315.7    6930  243.64    6930  8784.7   247.8
Permanent Ineff=
       F       F
Bank Sta=4949.5,5041.1
XS Rating Curve= 0 ,0
Exp/Cntr=0.3,0.1

Type RM Length L Ch R = 1 ,390222  ,4953,4953,4953
BEGIN DESCRIPTION:
NAVASOTA RIVER 397
END DESCRIPTION:
XS GIS Cut Line= 3
      3600937.82     10313984.65      3592880.24     10311762.41
      3587917.03     10310794.56
#Sta/Elev= 30
 -3358.4  292.45 -3186.5  291.31 -2765.2  244.52 -2553.4  244.76 -2350.7  240.12
  -244.7  240.69  -109.4  242.39  2289.4  239.38  2420.1  238.76  2619.4  237.87
  3217.5  239.16  3626.6  240.04  3795.2   240.4  4086.5  239.97  4378.3  240.26
  4948.9  242.68  4996.2  232.58  5130.1  242.58  5466.8  234.23  6914.8  235.15
  7379.2  244.11  7473.9  233.49  7514.6  242.23  8114.8  241.91  8400.3  242.31
  8560.5  243.87  8700.3  244.12  9261.9  247.66  9628.3  271.38 10056.7  315.57
#Mann= 20 ,-1 , 0
 -3358.4     .05       0 -2553.4     .16       0 -2350.7     .12       0
  -244.7     .07       0  -109.4     .12       0  2289.4     .12       0
  2420.1     .07       0  2619.4     .12       0  3217.5     .07       0
  3626.6     .12       0  3795.2     .07       0  4086.5     .07       0
  4378.3     .12       0  4948.9     .07       0  5130.1     .12       0
  8114.8     .16       0  8400.3     .16       0  8560.5     .12       0
  8700.3     .05       0  9261.9     .16       0
#XS Ineff= 2 , 0
       0                  7379.2       0  244.11
Permanent Ineff=
       F       F
Bank Sta=4948.9,5130.1
XS Rating Curve= 0 ,0
Exp/Cntr=0.3,0.1

Type RM Length L Ch R = 1 ,385269  ,2713,2713,2713
BEGIN DESCRIPTION:
NAVASOTA RIVER 398
END DESCRIPTION:
XS GIS Cut Line= 4
       3600048.6     10310756.57      3593824.64     10310157.61
      3592900.16     10309493.55       3586350.7     10309415.43
#Sta/Elev= 30
 -1609.5  290.28 -1322.5  277.59 -1123.3  267.27  -661.1  251.29   -25.7  237.91
   844.7  240.72   917.8  240.57  2993.6  237.72  3054.2  237.02  4354.4  240.12
  4557.2  233.87  4712.1  238.09  4950.7  239.93  5015.5  230.34  5042.8  240.34
  5051.4  240.65  7279.6  234.71  7389.6  241.16  8379.7  242.05  8409.7  232.13
  8459.7  231.93  8489.7  241.37   10219   238.7 10483.8  238.78 10696.1  238.88
 10794.8   239.7 11658.8  266.72 11948.4  293.62   12160  321.36 12331.4  323.11
#Mann= 18 ,-1 , 0
 -1609.5     .16       0 -1322.5     .12       0 -1123.3     .05       0
  -661.1     .12       0   844.7     .07       0   917.8     .12       0
  2993.6     .07       0  3054.2     .12       0  4557.2     .07       0
  4712.1     .12       0  4950.7     .07       0  5051.4     .12       0
   10219     .07       0 10483.8     .12       0 10696.1     .16       0
 10794.8     .05       0 11658.8     .16       0 11948.4     .05       0
#XS Ineff= 2 , 0
       0                  8379.7       0  242.05
Permanent Ineff=
       F       F
Bank Sta=4950.7,5042.8
XS Rating Curve= 0 ,0
Exp/Cntr=0.3,0.1

Type RM Length L Ch R = 1 ,382556  ,2777,2777,2777
BEGIN DESCRIPTION:
NAVASOTA RIVER 338
END DESCRIPTION:
XS GIS Cut Line= 3
      3597851.17     10308936.01        3594741.       10308151.
      3586525.43     10307935.37
#Sta/Elev= 30
  1792.3  292.81  2814.4  254.25  4147.1  259.17  4256.3  259.77    4383   251.7
  4658.5  232.33  4939.1  237.41  4979.9  229.56  5068.9  238.07  5127.6  237.45
  5355.6  239.09  5481.9  239.83  5613.4  240.37  6074.1  240.51  7298.3  238.69
  7690.4  238.19  8072.6  237.53  9010.3  240.47  9050.3   230.8  9100.3  239.19
    9291  239.75 10472.3  239.31 10614.9  238.86 11037.8  239.13 12094.8  247.78
 12193.5  252.59 12431.5  252.33   12458   257.4 12781.6  266.86 13218.4   307.9
#Mann= 20 ,-1 , 0
  1792.3     .05       0  4147.1     .16       0    4383     .12       0
  4939.1     .07       0  5068.9     .12       0  5127.6     .07       0
  5355.6     .12       0  5481.9     .07       0  5613.4     .12       0
  6074.1     .07       0  7298.3     .12       0  7690.4     .07       0
  8072.6     .12       0    9291     .12       0 10472.3     .05       0
 10614.9     .12       0 11037.8     .05       0 12094.8     .08       0
 12193.5     .05       0   12458     .16       0
#XS Ineff= 2 , 0
       0  4235.7  260.25  9010.3       0  240.47
Permanent Ineff=
       F       F
Bank Sta=4939.1,5068.9
XS Rating Curve= 0 ,0
Exp/Cntr=0.3,0.1

Type RM Length L Ch R = 1 ,379779  ,2736,2736,2736
BEGIN DESCRIPTION:
NAVASOTA RIVER 337
END DESCRIPTION:
XS GIS Cut Line= 3
      3597919.75     10308907.65      3593591.75     10306666.34
      3586352.16     10305650.71
#Sta/Elev= 30
  -398.1  293.99   495.1  257.05  1006.9  251.33  1948.3  258.13  2245.7  259.55
  2585.2  245.23  2694.2  238.28    2847   236.3  4057.5  238.78  4212.5  231.54
  4548.4   244.5  4576.4  233.73  4640.1  236.84  4739.3  236.79  4838.4  236.96
  4950.1  236.95  5010.4  226.95  5052.8   236.9  5119.1  228.79  5212.6  238.41
  5886.7  239.58  6102.4  240.76  6820.3  237.92  7025.2  237.97  8042.3  237.86
  8407.8  238.15 11392.5  266.04 11528.3   270.3 11707.6  301.15 11786.3  305.39
#Mann= 17 ,-1 , 0
  -398.1     .05       0  1948.3     .16       0  2585.2     .07       0
  2694.2     .12       0    2847     .05       0  4640.1     .12       0
  4739.3     .05       0  4838.4     .12       0  4950.1     .07       0
  5052.8     .12       0  5886.7     .16       0  6102.4     .12       0
  6820.3     .05       0  7025.2     .12       0  8042.3      .1       0
  8407.8     .05       0 11707.6     .16       0
#XS Ineff= 2 , 0
       0  2245.7  259.55               0
Permanent Ineff=
       F       F
Bank Sta=4950.1,5052.8
XS Rating Curve= 0 ,0
Exp/Cntr=0.3,0.1

Type RM Length L Ch R = 1 ,377043  ,2138,2138,2138
BEGIN DESCRIPTION:
NAVASOTA RIVER 336
END DESCRIPTION:
XS GIS Cut Line= 2
      3597992.66      10308756.6      3590941.12     10301715.36
#Sta/Elev= 30
    -547  293.84   977.2  250.59  1788.2  246.36  1819.5  246.25  4279.4  245.67
  4614.7  234.19  4697.1  237.72  4781.4  239.09  4852.1  229.63    4944  235.64
  5007.4  225.72  5050.1  239.98  5453.2  237.45  5481.4  231.88  5580.4  238.02
  5721.9  233.38  5905.7  238.13  6096.6  233.32    6132  237.64  7365.1  233.99
  7883.3  233.89  8054.8  238.96  8137.7  239.93  8253.3  241.29  8712.9  281.68
  9002.1  296.18  9032.6   297.9  9284.5  307.81    9407  304.29  9418.1     304
#Mann= 15 ,-1 , 0
    -547     .05       0  1788.2     .16       0  1819.5     .05       0
  4614.7     .12       0  4697.1     .05       0  4781.4     .07       0
  5050.1     .12       0  7365.1     .05       0  7883.3     .12       0
  8054.8     .05       0  8137.7     .16       0  9002.1     .05       0
  9032.6     .16       0  9284.5     .05       0    9407     .16       0
Bank Sta=4781.4,5050.1
XS Rating Curve= 0 ,0
Exp/Cntr=0.3,0.1

Type RM Length L Ch R = 1 ,374905  ,422,422,422
BEGIN DESCRIPTION:
NAVASOTA RIVER 335
END DESCRIPTION:
XS GIS Cut Line= 6
      3599449.48     10308886.23      3597451.86     10306729.39
      3595961.58     10305003.56      3594932.81     10303875.15
      3592674.95       10301438.      3591238.82     10299796.47
#Sta/Elev= 30
 -1189.7  291.49  -112.7  294.24   375.5  265.15  2001.8  260.33  2144.4  260.54
  2228.1  260.66  3168.5  262.29  3906.7  250.72  3995.6  237.69  4166.2   235.3
  4923.5  237.11  5029.5  227.95  5057.9  237.98  6409.4  235.45  6444.3  225.64
  6501.3  236.23  7513.6  231.17  8669.2  241.76  8862.4     254  9275.7  283.56
  9510.2  275.07  9545.3  266.12  9808.8  280.48  9926.7  285.44 10162.2  295.07
 10357.3  289.12 10484.5  289.57 10500.9  289.75 10754.8     298 11060.8  297.48
#Mann= 19 ,-1 , 0
 -1189.7     .05       0  2001.8     .08       0  2144.4      .1       0
  2228.1     .05       0  3906.7     .12       0  4923.5     .07       0
  5057.9     .12       0  6409.4     .07       0  6501.3     .12       0
  8669.2     .16       0  8862.4     .05       0  9808.8     .16       0
  9926.7     .05       0 10357.3     .05       0 10357.3     .16       0
 10484.5     .05       0 10500.9     .16       0 10754.8     .05       0
 11060.8     .05       0
Bank Sta=4923.5,5057.9
XS Rating Curve= 0 ,0
Exp/Cntr=0.3,0.1

Type RM Length L Ch R = 1 ,374483  ,4944,4944,4944
BEGIN DESCRIPTION:
NAVASOTA RIVER 334
END DESCRIPTION:
XS GIS Cut Line= 6
       3599735.6     10308621.21      3597740.95     10306467.57
      3595954.58     10304412.79      3592964.76     10301176.96
      3592123.83     10300182.21      3591641.05     10299521.77
#Sta/Elev= 30
 -1315.1  289.54  -223.4  291.24   454.2  271.32  1730.1  251.82  1871.4  259.92
  3154.6  260.44  3670.5  244.66  4132.6  235.86  4600.3  236.77  4940.4  237.48
  4975.6  227.17    5110  233.72  5294.5  227.47  5336.4  237.95  5818.3  236.67
    5989  234.71  6291.9  238.49  6369.3  225.57  6447.3  239.31  6960.3  233.96
  7350.3  234.25  7516.3  234.81  8308.6  233.55  8626.8  248.42  9002.7  277.35
  9308.3  267.37  9452.8  271.37  9863.7  286.27 10090.8  292.95 10869.9  297.01
#Mann= 19 ,-1 , 0
 -1315.1     .05       0   454.2     .05       0  3670.5     .12       0
  4132.6     .12       0  4600.3     .12       0  4940.4     .07       0
  5336.4     .12       0  5818.3     .12       0    5989     .12       0
  6291.9     .07       0  6447.3     .07       0  6960.3     .12       0
  7350.3     .12       0  7516.3     .12       0  8626.8     .05       0
  9308.3     .16       0  9452.8     .05       0  9863.7     .05       0
 10090.8     .05       0
Bank Sta=4940.4,5336.4
XS Rating Curve= 0 ,0
Exp/Cntr=0.3,0.1

Type RM Length L Ch R = 1 ,369539  ,3458,3458,3458
BEGIN DESCRIPTION:
NAVASOTA RIVER 405
END DESCRIPTION:
XS GIS Cut Line= 3
      3599848.49     10305545.51      3597454.62     10303436.01
      3592405.99     10299322.93
#Sta/Elev= 30
  1809.3  293.21  2057.7  285.66  2259.7  268.33  2574.9  248.65  2898.3  241.54
  3026.6  238.98  3182.1  238.47  3534.5  236.36  3936.1  234.88    4298  235.36
  4962.7  236.46  4990.3  226.31  5076.2  236.14    6985  235.18    7769  235.95
  8033.4  236.54  8086.4  225.68  8089.1  225.18  8092.4  225.68  8263.4  234.07
  8771.6  228.85  8878.6  247.77  8971.1  241.14  9503.5  241.08  9731.1  246.69
 10087.2  271.57 10321.3  263.39 10737.9  270.02 11316.6  298.15   11512  296.13
#Mann= 20 ,-1 , 0
  1809.3     .05       0  2259.7     .05       0  2898.3     .05       0
  3026.6     .05       0  3182.1     .07       0  3534.5     .12       0
  3936.1     .12       0    4298     .12       0  4962.7     .07       0
  5076.2     .12       0    6985     .12       0    7769     .12       0
  8086.4     .07       0  8092.4     .07       0  8263.4     .12       0
  8971.1     .05       0  9503.5     .12       0  9731.1     .16       0
 10087.2     .05       0 10737.9     .05       0
Bank Sta=4962.7,5076.2
XS Rating Curve= 0 ,0
Exp/Cntr=0.3,0.1

Type RM Length L Ch R = 1 ,366081  ,3637,3637,3637
BEGIN DESCRIPTION:
NAVASOTA RIVER 408
END DESCRIPTION:
XS GIS Cut Line= 3
      3601071.69     10304246.23       3598359.8     10302085.71
      3592296.37     10298890.71
#Sta/Elev= 30
  1532.7  291.23  1899.7  271.26    2351  239.05  4965.8  234.86  4986.6  225.77
  5066.6  234.52  5121.4  234.77    6102  234.89  6517.4  235.04  6675.6  234.81
  6871.5  234.53  7180.6  233.16  7321.3  233.69    7518  237.38  7554.2  225.72
  7633.6  225.68  7636.4  225.18  7639.6  225.68  7746.4  235.64  7785.2  235.87
  7829.2  251.45    7889  241.09    9387   241.3  9605.8  241.01  9948.3  268.84
 10146.2  277.79 10278.4  265.47 10773.7  263.67 11035.6  276.27 11853.7  294.02
#Mann= 20 ,-1 , 0
  1532.7     .05       0  1899.7     .16       0    2351     .12       0
  4965.8     .07       0  4965.8     .07       0  5121.4     .12       0
    6102     .16       0  6517.4     .16       0  6675.6      .1       0
  6871.5     .05       0  7180.6     .05       0  7321.3     .05       0
  7633.6     .07       0  7639.6     .05       0  7746.4     .12       0
    7889     .05       0    9387     .07       0  9605.8     .12       0
  9948.3     .05       0 11035.6     .05       0
Bank Sta=4965.8,5066.6
XS Rating Curve= 0 ,0
Exp/Cntr=0.3,0.1

Type RM Length L Ch R = 1 ,362444  ,3051,3051,3051
BEGIN DESCRIPTION:
NAVASOTA RIVER 407
END DESCRIPTION:
XS GIS Cut Line= 3
      3603816.71     10302637.81      3599971.78     10300443.53
      3592235.68     10298678.93
#Sta/Elev= 30
     573  285.33   637.7  285.02   748.9  283.05   853.3  284.49  1209.2     252
    1558  240.33  1653.4  238.32  3917.3  229.84  4913.1  233.99  5028.1  226.02
  5081.7  235.09  7666.4  236.07  7707.5  225.96  7830.3  225.34  7892.1  236.18
  8302.4  232.54  8391.5     239  8491.9  238.89  8692.7  233.75  9695.1  234.36
  9953.7  248.58 10021.3  241.65 10245.8  244.97 10523.3  246.18 10579.4  241.45
 10961.9  250.77 11072.4  250.45 11329.8  253.01 11605.1  272.33 12934.8  292.78
#Mann= 19 ,-1 , 0
     573      .1       0   637.7     .15       0   748.9     .16       0
  1209.2     .12       0    1558     .05       0  1653.4     .12       0
  4913.1     .07       0  5081.7     .12       0  7666.4     .07       0
  7666.4     .07       0  7892.1     .12       0  8391.5     .15       0
  8491.9      .1       0  8692.7     .12       0  9695.1     .05       0
 10245.8     .16       0 10523.3     .05       0 10961.9     .16       0
 11072.4     .05       0
Bank Sta=4913.1,5081.7
XS Rating Curve= 0 ,0
Exp/Cntr=0.3,0.1

Type RM Length L Ch R = 1 ,359393  ,2718,2718,2718
BEGIN DESCRIPTION:
NAVASOTA RIVER 193
END DESCRIPTION:
XS GIS Cut Line= 3
      3604583.95      10301898.8      3599913.78     10298999.48
      3592136.54     10298391.88
#Sta/Elev= 30
    37.4   277.7    40.5  277.66   270.8  279.83   384.3  263.17   611.2  258.27
     784  232.61   814.7  239.97  4952.8  233.89  5004.6  224.03  5041.4  232.77
    5923  234.07  6293.9  234.04  6853.5  232.95    6950  232.76  7090.8  235.03
    7161  225.59  7191.1  235.96  7311.4  230.05  8010.3   233.8  8363.6  233.95
  8854.5  234.58  9150.8  236.07  9842.1  232.69  9940.9  244.31 10039.6  244.52
 10245.5  236.17 10434.7   240.5 11990.5  248.87 12886.2  283.35 13335.3  287.96
#Mann= 20 ,-1 , 0
    37.4     .12       0    40.5     .16       0   270.8     .08       0
   384.3     .05       0   611.2     .12       0  4952.8     .07       0
  5041.4     .12       0    5923     .05       0  6293.9     .05       0
  6853.5     .07       0    6950     .12       0  8010.3     .12       0
  8363.6     .05       0  8854.5      .1       0  9150.8     .05       0
  9842.1      .1       0  9940.9     .08       0 10039.6     .05       0
 10245.5     .16       0 10434.7     .05       0
Bank Sta=4952.8,5041.4
XS Rating Curve= 0 ,0
Exp/Cntr=0.3,0.1

Type RM Length L Ch R = 1 ,356675  ,3973,3973,3973
BEGIN DESCRIPTION:
NAVASOTA RIVER 406
END DESCRIPTION:
XS GIS Cut Line= 3
       3607947.8     10298250.65      3601399.73     10298095.53
      3590755.11     10297665.65
#Sta/Elev= 30
 -1549.9  288.77 -1477.4  287.98    -804  246.84  -227.4  240.87   347.3  238.12
   605.4  242.06   906.5  250.41  1180.8  239.04  1674.3  235.79  2365.2  237.64
  3118.5  236.47  4847.6  233.46  5007.4  223.54  5047.7  233.18  5720.9  234.61
  6016.9  234.38  6625.4  233.32  7168.2  232.71  7398.5  232.45  7793.3  232.83
  8429.4  232.42  8615.1  232.07 10063.1  236.77 13124.2     243 13694.7  264.31
   14015  262.12 14285.2  282.79 14475.3  271.24   15246  271.74 15653.3  293.24
#Mann= 20 ,-1 , 0
 -1549.9     .05       0 -1477.4     .16       0  -227.4     .05       0
   347.3     .05       0   605.4     .16       0  1180.8     .12       0
  1674.3     .05       0  2365.2     .12       0  3118.5     .12       0
  4847.6     .07       0  5047.7     .12       0  5720.9     .16       0
  6016.9     .05       0  6625.4     .12       0  7168.2      .1       0
  7398.5     .05       0  7793.3     .12       0  8429.4     .07       0
  8615.1     .12       0 10063.1     .05       0
#XS Ineff= 4 ,-1
  -958.8   906.5  250.41   906.5    2687  237.98    2687  3027.1  237.52
  3027.1  4027.4  235.06
Permanent Ineff=
       F       F       F       F
Bank Sta=4847.6,5047.7
XS Rating Curve= 0 ,0
Exp/Cntr=0.3,0.1

Type RM Length L Ch R = 1 ,352702  ,3139,3139,3139
BEGIN DESCRIPTION:
NAVASOTA RIVER 403
END DESCRIPTION:
XS GIS Cut Line= 3
      3608025.17     10296998.65      3601667.96     10296230.08
      3590657.18     10296386.64
#Sta/Elev= 30
 -1403.5  284.41 -1166.9  280.86  -884.3  274.61  -639.9  250.44    -418  241.53
    77.1  237.62  1314.4  234.82  2350.6  232.76  3655.2  231.55  4488.2  232.74
  4947.9  232.44  4995.1   223.5  5045.9  233.45  5558.6  233.21  6608.8  231.28
  6955.2  231.03  7881.6  231.31  8146.2  233.48  8188.3   225.2  8964.7  232.83
  9573.6  235.34 10006.4  239.54 10226.4  231.21 10269.9  237.06 11154.8  235.99
 11757.3  236.83 15206.9  246.11 15566.9   255.2   15827  280.02 16011.9  280.79
#Mann= 20 ,-1 , 0
 -1403.5     .05       0 -1166.9     .16       0    -418     .12       0
    77.1     .05       0  1314.4     .05       0  2350.6     .07       0
  3655.2     .07       0  4488.2     .12       0  4947.9     .07       0
  5045.9     .12       0  5558.6     .16       0  6608.8     .12       0
  6955.2     .05       0  7881.6     .05       0  8188.3     .12       0
  8964.7     .12       0  9573.6     .16       0 10269.9     .16       0
 11154.8     .16       0 11757.3     .05       0
#XS Ineff= 4 ,-1
  8146.2  9681.5  233.48  9681.5 10766.4  238.76 10766.4 13846.8  240.88
  -474.5  1358.6  237.07
Permanent Ineff=
       F       F       F       F
Bank Sta=4947.9,5045.9
XS Rating Curve= 0 ,0
Exp/Cntr=0.3,0.1

Type RM Length L Ch R = 1 ,349563  ,1698,1698,1698
BEGIN DESCRIPTION:
NAVASOTA RIVER 404
END DESCRIPTION:
XS GIS Cut Line= 4
      3608084.33     10296563.92       3601321.8     10294529.56
      3591463.91     10295428.16      3590975.67     10295734.61
#Sta/Elev= 30
 -2061.9  283.38 -1921.3  280.82 -1590.1  274.78 -1411.6  261.24   -1173  241.85
 -1003.9  242.24  -196.4  235.33   164.7  245.63  1034.7   232.8  1959.1  232.36
  3258.2   231.3  3809.2  226.03  3984.2  231.69  4122.5  225.71  4694.7  231.37
  4947.5  230.26    4997  222.14  5049.9  231.79  5109.3  231.61    5806  229.53
  7000.3  230.71  7398.4  231.36  8294.1  231.88    8846  233.35 10350.4  234.65
 11939.7  236.89   12324   236.7 14097.3  235.06 14883.8  274.61 15475.2  281.19
#Mann= 20 ,-1 , 0
 -2061.9     .05       0 -1921.3     .16       0 -1411.6     .12       0
 -1003.9     .05       0  -196.4     .16       0  1034.7     .05       0
  1959.1     .07       0  3258.2     .12       0  3984.2     .12       0
  4694.7     .07       0  5049.9     .12       0  5109.3      .1       0
    5806     .12       0  7000.3     .05       0  7398.4     .12       0
  8294.1     .16       0    8846     .16       0 10350.4     .05       0
 11939.7     .16       0   12324     .05       0
#XS Ineff= 2 , 0
       0   164.7  245.63 11345.9       0  239.65
Permanent Ineff=
       F       F
Bank Sta=4694.7,5049.9
XS Rating Curve= 0 ,0
Exp/Cntr=0.3,0.1

Type RM Length L Ch R = 1 ,347865  ,1230,1230,1230
BEGIN DESCRIPTION:
NAVASOTA RIVER 402
END DESCRIPTION:
XS GIS Cut Line= 3
      3608151.03     10296493.88      3603705.71     10293273.39
      3593789.09     10293186.58
#Sta/Elev= 30
 -3174.9  283.79 -2934.5  276.81 -2636.6  279.18 -2364.3  250.17 -2236.9  238.28
 -2046.7  240.27 -1013.7  238.47  -562.8  237.83  1489.4  235.36    3388  226.63
  4948.1   231.6  4998.1  223.79  5048.1  231.92  5388.1  231.57  5408.1  223.72
  5527.9  222.24  5588.1  231.64  5818.1  231.12  5868.1  223.37  5888.1  231.06
  5941.5  229.35  6549.1  230.77  7464.1  230.82  7669.9  231.23    8083  232.05
  8469.5  232.81  9256.9  233.43 11584.9   235.2 11869.1  246.86 12231.4  270.08
#Mann= 20 ,-1 , 0
 -3174.9     .05       0 -2934.5     .16       0 -2364.3     .16       0
 -2046.7     .05       0 -1013.7     .16       0  -562.8     .05       0
  1489.4     .12       0  4948.1     .07       0  5048.1     .12       0
  5388.1     .07       0  5588.1     .12       0  5941.5     .07       0
  6549.1     .12       0  7464.1     .12       0  7669.9     .16       0
    8083     .12       0  8469.5     .16       0  9256.9     .05       0
 11584.9     .05       0 11869.1     .16       0
#XS Ineff= 3 ,-1
  5388.1  5658.1  231.57  5658.1  8469.5  232.48 10878.3 11869.1  237.09
Permanent Ineff=
       F       F       F
Bank Sta=4948.1,5048.1
XS Rating Curve= 0 ,0
Exp/Cntr=0.3,0.1

Type RM Length L Ch R = 1 ,346635  ,911,911,911
BEGIN DESCRIPTION:
NAVASOTA RIVER 194
END DESCRIPTION:
XS GIS Cut Line= 4
      3606703.35     10292277.47      3601141.84     10292128.93
      3598333.92     10292055.04      3593299.17     10291707.81
#Sta/Elev= 30
  -563.5  284.88  -157.6  271.78     248  234.02   592.1  230.59  1828.6  234.62
  2528.8  231.98  2638.9  226.79  2668.9  231.29  4959.7   231.4  4997.4  223.68
  5085.8  229.55  5259.8  231.22  5319.8  228.16  5529.9  231.51  5589.9   225.7
    5710  228.64    5780  225.26    5820  231.25  6030.1  230.57  6089.9  221.28
  6150.1   223.1  6180.1  230.77  6413.4   230.5  6460.8  230.45  8431.8  232.72
  8843.2  231.82  9345.5  232.38 11679.9  233.89 12391.6  284.05 12855.6  263.55
#Mann= 10 ,-1 , 0
  -563.5     .16       0  4959.7     .07       0  5259.8     .12       0
  6030.1     .07       0  6180.1     .12       0  6413.4     .07       0
  6460.8     .12       0  8431.8     .05       0  8843.2     .12       0
  9345.5     .05       0
#XS Ineff= 3 ,-1
  5509.9  8422.2  231.73  9594.9 11840.3  235.35  8422.2  9594.9  232.84
Permanent Ineff=
       F       F       F
Bank Sta=4959.7,5259.8
XS Rating Curve= 0 ,0
Exp/Cntr=0.3,0.1

Type RM Length L Ch R = 1 ,345724  ,2335,2335,2335
BEGIN DESCRIPTION:
NAVASOTA RIVER 195
END DESCRIPTION:
XS GIS Cut Line= 3
      3605878.79     10291088.58      3602431.14     10291499.48
       3593368.6     10289884.89
#Sta/Elev= 30
   488.3  281.98   669.1  277.01  1028.1  239.98  1211.7  230.36  1367.2  231.69
  4934.5  230.69  5006.5     220    5097  230.31  5452.5  231.38  5493.2  222.42
    5615   230.6    6194  224.33  6317.5  231.18  6417.5  222.79  6510.1  229.03
  6710.1  230.07  8116.3  230.25  8350.4  230.71    8655  230.88    8802   230.9
 10507.9  231.81 10716.1  231.28 11067.1   230.4 11469.3   230.6 12191.3  241.75
 12645.8  281.93 12803.8  279.53 12897.9  273.01   13015  285.32 13165.6  299.67
#Mann= 20 ,-1 , 0
   488.3     .12       0   669.1     .16       0  1028.1     .12       0
  1211.7     .16       0  1367.2     .12       0  4934.5     .07       0
    5097     .12       0  6510.1     .07       0  6710.1     .12       0
  8116.3     .05       0  8350.4     .12       0    8655     .05       0
    8802     .12       0 10507.9     .05       0 10716.1     .07       0
 11067.1     .12       0 11469.3     .05       0 12191.3     .05       0
 12803.8     .16       0   13015     .05       0
Bank Sta=4934.5,5097
XS Rating Curve= 0 ,0
Exp/Cntr=0.3,0.1

Type RM Length L Ch R = 1 ,343389  ,2572,2572,2572
BEGIN DESCRIPTION:
NAVASOTA RIVER 196
END DESCRIPTION:
XS GIS Cut Line= 4
      3605283.04     10289422.63      3602579.41     10289784.19
      3602257.53     10289832.81      3594515.81     10287992.85
#Sta/Elev= 30
  2272.3  257.53    2297  257.13  2529.7   244.9  2646.5  249.45  2745.8  237.39
  3027.9   240.1  3212.2  232.76  3776.5  229.79  3857.2  225.15  3877.4  229.07
  4079.2  224.04  4210.3  229.27  4956.9  230.19  4977.1  221.15  5007.1  218.91
  5118.6  229.12  7191.5  230.13  7232.6  220.15  7346.2  229.37  7499.9  230.14
  7941.9  225.13  8404.4  230.26 10181.4  229.81 10480.5  229.56   11883  230.86
 12578.6  262.13 12865.3  265.04 12978.3   261.1 13137.2  270.23 13282.9   270.8
#Mann= 9 ,-1 , 0
  2272.3     .16       0    2297     .12       0  2745.8     .16       0
  3027.9     .12       0  4956.9     .07       0  5118.6     .12       0
 10181.4     .16       0 10480.5     .12       0   11883     .16       0
Bank Sta=4956.9,5118.6
XS Rating Curve= 0 ,0
Exp/Cntr=0.3,0.1

Type RM Length L Ch R = 1 ,340817  ,2893,2893,2893
BEGIN DESCRIPTION:
NAVASOTA RIVER 197
END DESCRIPTION:
XS GIS Cut Line= 4
      3604030.34     10287933.87      3602902.46      10288004.7
      3600608.22     10288148.79      3595486.91     10286985.64
#Sta/Elev= 30
  3869.9   249.2  4089.2  234.08  4228.5  220.12    4329  228.18  4539.4  228.63
  4599.6  222.69  4713.3  229.03  4930.2  228.19  4960.3  220.04  5020.1   217.9
  5070.5  228.36  7533.3  229.71  7633.7  229.68  7746.2  229.57  7831.4  229.51
  8155.7  229.98  8209.9  226.61  8303.3  221.46  8523.9  229.93  9071.6  225.59
 10835.8  230.55   11243  257.45 11307.9  262.61 11602.3  283.58 11918.3  291.97
   12251  286.84 12339.4  285.78 12351.4  285.72 12451.8  285.22 12550.5   284.9
#Mann= 18 ,-1 , 0
  3869.9     .05       0  4089.2     .12       0  4930.2     .07       0
  5070.5     .12       0  7533.3     .07       0  7633.7     .12       0
  7746.2     .07       0  7831.4     .12       0  8155.7     .07       0
  8209.9     .12       0 10835.8     .16       0   11243     .05       0
 11307.9     .16       0 11918.3     .05       0   12251      .1       0
 12339.4     .05       0 12351.4      .1       0 12451.8     .16       0
Bank Sta=4930.2,5070.5
XS Rating Curve= 0 ,0
Exp/Cntr=0.3,0.1

Type RM Length L Ch R = 1 ,337924  ,2643,2643,2643
BEGIN DESCRIPTION:
NAVASOTA RIVER 198
END DESCRIPTION:
XS GIS Cut Line= 3
      3603681.14     10285891.84      3602014.47     10286291.15
      3595556.65     10286065.47
#Sta/Elev= 30
    4262  254.37  4611.4  256.04  4826.6  256.52  4891.6   252.3  4919.1  248.45
    4931   240.2    4950  228.22  4990.8  216.62  5042.5  219.21  5063.1  228.17
  6338.4  225.23  7479.1  229.06  7569.2  220.45  7609.2   224.4  7639.2  219.82
  7709.3  228.83  8125.4  227.95  8130.8  227.96  9018.9  228.37  9120.9  228.29
  9524.1   230.2  9703.5  230.72  9907.1   231.3 10557.7  231.83 10755.3  231.63
 11614.2  235.15 11861.8  236.81   12132   246.5 12358.3  262.59 12437.6  266.13
#Mann= 17 ,-1 , 0
    4262     .16       0  4611.4     .05       0  4891.6     .16       0
    4931     .12       0    4950     .07       0  5063.1     .12       0
  8125.4     .07       0  8130.8     .12       0  9018.9     .05       0
  9120.9     .12       0  9524.1     .16       0  9703.5     .12       0
  9907.1     .05       0 10557.7     .07       0 10755.3     .05       0
 11614.2     .16       0 12358.3     .05       0
Bank Sta=4950,5063.1
XS Rating Curve= 0 ,0
Exp/Cntr=0.3,0.1

Type RM Length L Ch R = 1 ,335281  ,2092,2092,2092
BEGIN DESCRIPTION:
NAVASOTA RIVER 401
END DESCRIPTION:
XS GIS Cut Line= 5
       3605276.4     10286294.37      3602607.11     10285044.37
      3602437.84     10284436.73      3601417.01     10284465.37
      3595192.19     10285819.54
#Sta/Elev= 30
  1318.5  268.77  1411.5  266.19  1484.8  264.16  1532.6  262.65  1690.3   255.6
    2153  248.13  2322.7  249.11  2495.9  241.65  2558.7  241.53  2581.5  247.65
  2655.5  252.58  2930.6  252.33  4292.8  252.68  4677.4  246.09  4896.8  229.91
  4942.5  225.86  4982.3  214.17  5022.5  217.29  5042.5  224.32  5132.6  228.21
  5412.7  228.89  5732.8  219.65  5842.9  226.84  7294.3  225.39  8409.8   233.8
  9369.3  233.84 11514.8  239.05 11797.3  242.96   12053  256.45 12288.4  270.31
#Mann= 15 ,-1 , 0
  1318.5     .05       0  1411.5      .1       0  1484.8     .05       0
  1532.6     .16       0  1690.3     .05       0    2153     .16       0
  2322.7     .05       0  2495.9     .16       0  2930.6     .05       0
  4292.8     .12       0  4896.8     .07       0  5132.6     .12       0
  9369.3     .05       0 11514.8     .16       0   12053     .05       0
#XS Ineff= 2 , 0
       0  3693.2  254.85  8607.4       0  234.46
Permanent Ineff=
       F       F
Bank Sta=4896.8,5132.6
XS Rating Curve= 0 ,0
Exp/Cntr=0.3,0.1

Type RM Length L Ch R = 1 ,333189  ,102,102,102
BEGIN DESCRIPTION:
NAVASOTA RIVER 399
END DESCRIPTION:
XS GIS Cut Line= 6
      3607124.92     10285813.28      3603105.45     10284863.12
      3601846.22     10283050.22      3598940.68     10284342.54
      3597967.77     10284208.49      3595890.73     10283155.46
#Sta/Elev= 30
 -1746.9  266.28 -1707.6  266.28   -97.1  251.37   808.4   250.6  1513.5  250.46
  2419.6  251.26  2697.9  250.06  2955.1  242.44  3243.3  226.04  3630.5  224.75
  4630.6   221.9  4861.4  227.62  4947.1  228.13  4968.1  221.64  5080.1  220.49
  5180.8  228.64  5543.3  222.35  5800.9   227.6  6101.1  229.05    6205  221.46
  6257.5   229.7  6642.4     227  7097.4  229.69  7418.2  231.89    7689  232.58
  8225.8  232.87  9376.1  232.98   10496  234.77 10934.3  245.66 11276.3  278.54
#Mann= 20 ,-1 , 0
 -1746.9     .16       0 -1707.6     .05       0   -97.1     .05       0
   808.4     .05       0  1513.5     .05       0  2419.6     .05       0
  2697.9     .05       0  2955.1     .05       0  3630.5     .05       0
  4861.4     .08       0  4947.1     .07       0  5180.8     .08       0
  5800.9     .12       0  6642.4     .08       0  7097.4     .05       0
  7418.2     .05       0    7689     .12       0  8225.8     .05       0
  9376.1     .05       0   10496     .05       0
#XS Ineff= 2 ,-1
  5961.6  8498.6  230.64  8498.6 10814.9  235.51
Permanent Ineff=
       F       F
Bank Sta=4947.1,5180.8
XS Rating Curve= 0 ,0
Exp/Cntr=0.3,0.1

Type RM Length L Ch R = 1 ,333087  ,1411,1411,1411
BEGIN DESCRIPTION:
NAVASOTA RIVER 400
END DESCRIPTION:
XS GIS Cut Line= 6
      3607143.31     10285727.37      3603146.36     10284771.46
      3601874.92     10282954.12      3600230.19     10283408.82
       3598928.9     10284242.54      3595858.77     10283054.21
#Sta/Elev= 30
 -1817.9  266.64 -1762.3  266.22    -352  252.86   376.6  244.78   719.1  248.62
  1459.9  251.71  1725.6  251.06  2680.2  250.09  3073.6  228.25  3504.6  225.61
  4397.6  229.84  4470.9  228.59  4492.3  221.67  4556.4  221.86    4578  229.41
  4843.8  229.61  5032.9  220.67  5074.9  229.41  5777.5  225.22  6978.6  227.59
  7082.4  233.37    7335   231.4  8159.6  233.01  8869.7  230.68  9545.3  232.31
  9761.6  233.05 10356.3  233.94 10870.8  246.45 11181.6  277.92 11258.8  281.79
#Mann= 20 ,-1 , 0
 -1817.9     .08       0 -1762.3     .05       0    -352     .05       0
   719.1     .05       0  1459.9     .05       0  1725.6     .16       0
  2680.2     .05       0  3504.6     .12       0  4397.6     .08       0
  4843.8     .07       0  5074.9     .12       0  5777.5     .05       0
  6978.6     .05       0    7335     .05       0  8159.6     .05       0
  8869.7     .05       0  9545.3     .08       0  9761.6     .05       0
 10356.3     .05       0 11181.6     .08       0
#XS Ineff= 2 ,-1
  5665.7  7082.4  229.71  7082.4 10616.4  233.37
Permanent Ineff=
       F       F
Bank Sta=4843.8,5074.9
XS Rating Curve= 0 ,0
Exp/Cntr=0.3,0.1

Type RM Length L Ch R = 1 ,331676  ,2269,2269,2269
BEGIN DESCRIPTION:
NAVASOTA RIVER 409
END DESCRIPTION:
XS GIS Cut Line= 4
      3605158.25     10283909.37      3601406.83     10282059.38
      3600970.15     10281988.95      3596938.24     10281224.73
#Sta/Elev= 30
   374.9     252   392.8  251.19   687.1   248.6     841  247.72  1328.1  232.18
  1558.4  225.54  1848.7  225.88  1965.5  226.01  2325.7  226.43  2593.4   226.6
  3325.6  229.85  3381.1  221.44  3415.4  228.75    3814  228.17  3931.9  221.31
  4044.2   230.1  4150.4  223.23    4195  229.68  4937.2  226.96  4987.6  220.56
  5059.1  226.82  5933.7  226.02  6162.7  226.22  6700.4  227.31  7163.4  228.46
    8148  229.49  8247.8  230.97  8447.3  235.34  8547.1  237.53  9103.7  272.91
#Mann= 20 ,-1 , 0
   374.9     .05       0   392.8     .16       0   687.1     .05       0
     841     .16       0  1328.1     .12       0  1558.4     .05       0
  1848.7     .12       0  1965.5     .12       0  2325.7     .16       0
  2593.4     .12       0  4937.2     .07       0  5059.1     .12       0
  5933.7     .16       0  6162.7     .12       0  6700.4     .05       0
  7163.4     .05       0    8148     .16       0  8247.8     .12       0
  8447.3      .1       0  8547.1     .05       0
#XS Ineff= 2 , 0
       0                  5130.3       0  227.69
Permanent Ineff=
       F       F
Bank Sta=4937.2,5059.1
XS Rating Curve= 0 ,0
Exp/Cntr=0.3,0.1

Type RM Length L Ch R = 1 ,329407  ,1755,1755,1755
BEGIN DESCRIPTION:
NAVASOTA RIVER 199
END DESCRIPTION:
XS GIS Cut Line= 3
      3603727.74     10279821.73      3600456.31     10279963.02
      3596876.34     10279702.66
#Sta/Elev= 30
  2362.6  244.41  2848.7  244.32  3058.9  237.19  3249.1  240.95  3413.6  224.07
  3512.6  223.45  3611.7  222.27  3799.6  226.57  3899.7  221.85  3949.7  225.62
    4220  221.27    4250  226.82  4345.4  226.22  4638.8  224.61  4940.6  225.62
  4980.4  220.54  5060.7  226.59    5999  225.27  6132.6  221.46  6182.7  225.73
  6327.7  225.22  6579.4  224.64  7270.5  225.62  7566.7  227.02  8018.3  232.91
  8209.8  238.32  8508.8  257.15  8869.8  254.42  9080.3   263.3  9226.5  263.83
#Mann= 13 ,-1 , 0
  2362.6     .16       0  3413.6     .12       0  3512.6     .05       0
  3611.7     .12       0  4345.4     .07       0  4638.8     .12       0
  4940.6     .07       0  5060.7     .12       0  6327.7      .1       0
  6579.4     .05       0  7270.5     .16       0  7566.7     .05       0
  8018.3     .16       0
Bank Sta=4940.6,5060.7
XS Rating Curve= 0 ,0
Exp/Cntr=0.3,0.1
