HEC-RAS study NAVASOTA RIVER.prj: NAVASOTA RIVER Base Level Engineering

--- NAVASOTA RIVER.g01 (geometry) --- (continued)

Type RM Length L Ch R = 1 ,180103  ,1711,1711,1711
BEGIN DESCRIPTION:
NAVASOTA RIVER 273
END DESCRIPTION:
XS GIS Cut Line= 3
      3613471.58     10197031.71      3609420.73     10194989.76
      3604806.63     10191827.91
#Sta/Elev= 30
   463.6  252.34   583.3  251.83   884.8  223.76  1267.2  201.12  1375.6  198.18
  1587.1  199.22  1795.6  188.83  2876.7  188.44  3116.2   189.2  3265.7  183.75
  3326.8  189.98  4085.6  189.45  4302.4   189.3  4529.9  190.06  4646.5  189.57
  4871.7  191.87  5010.8  179.58  5091.6  192.01  5418.9  191.09  5531.9  190.77
  5874.8  185.91  6727.9  189.75  7047.1  214.28  8196.7  210.57  8679.7  216.98
  9521.4  215.39  9802.3  235.64 10077.2  232.26 10309.6  238.76 10593.5  240.27
#Mann= 20 ,-1 , 0
   463.6     .16       0   884.8     .05       0  1267.2     .16       0
  1375.6     .16       0  2876.7     .12       0  3116.2     .07       0
  3265.7     .07       0  3326.8     .05       0  4085.6     .07       0
  4302.4     .07       0  4529.9     .12       0  4646.5     .12       0
  4871.7     .07       0  5091.6     .12       0  5418.9     .07       0
  5531.9     .12       0  6727.9     .16       0  8196.7     .05       0
  8679.7     .16       0 10309.6     .05       0
#XS Ineff= 2 , 0
       0 3316.17  189.97  7277.4       0  216.17
Permanent Ineff=
       F       F
Bank Sta=4871.7,5091.6
XS Rating Curve= 0 ,0
Exp/Cntr=0.3,0.1

Type RM Length L Ch R = 1 ,178392  ,1299,1299,1299
BEGIN DESCRIPTION:
NAVASOTA RIVER 275
END DESCRIPTION:
XS GIS Cut Line= 3
      3615105.66     10195868.51      3609260.14     10193764.93
      3604808.36     10191738.73
#Sta/Elev= 30
 -1212.5  252.13 -1154.9  252.68  -944.8  250.33  -273.5  220.74   -86.1  196.11
   265.4  193.14  1915.9  183.49  2977.7  189.44  3147.5  189.46  3317.5  189.48
  3598.4  189.51  3818.4  189.54  4070.2  189.57  4425.9  189.62  4937.7  189.93
    4987  179.47  5052.8  189.58  5119.2  188.86    5680  188.47  5936.2  189.31
  6113.5  208.58    6225  217.24  7418.1  209.95    8045  212.13    8119  212.52
  8617.5  214.86    8859  231.41  9183.9  239.78  9629.7  240.01  9891.2  240.17
#Mann= 20 ,-1 , 0
 -1212.5     .05       0 -1154.9     .16       0   265.4     .12       0
  2977.7     .07       0  3147.5     .07       0  3317.5     .05       0
  3598.4     .12       0  3818.4     .07       0  4070.2     .05       0
  4425.9     .12       0  4937.7     .07       0  5052.8     .12       0
  5119.2     .12       0    5680     .12       0  5936.2     .16       0
  6113.5     .16       0  7418.1     .05       0    8045     .05       0
    8119     .16       0  9629.7     .05       0
#XS Ineff= 2 , 0
       0 2246.09  189.37    6225       0  217.24
Permanent Ineff=
       F       F
Bank Sta=4937.7,5052.8
XS Rating Curve= 0 ,0
Exp/Cntr=0.3,0.1

Type RM Length L Ch R = 1 ,177093  ,1714,1714,1714
BEGIN DESCRIPTION:
NAVASOTA RIVER 276
END DESCRIPTION:
XS GIS Cut Line= 3
      3615825.75     10194040.83      3609491.04     10192568.75
      3604758.13     10191612.27
#Sta/Elev= 30
 -1503.5  268.69 -1170.9  264.74  -893.5  232.68  -793.1  227.93    -586  219.73
  -202.4  228.95   276.3  223.28  1154.2  191.65  1364.6  183.32  3088.4   186.8
  3208.4   186.7  3569.2  186.85  3944.6  188.73  4921.4  190.24  4988.4  179.93
  5058.1  189.78  5930.6  188.72  6220.2  214.14    6630  215.64    6934     210
  7129.6  208.56  7429.3  216.82  7663.3  216.37  8194.2  214.92  8742.2  238.38
  9327.7   239.2  9427.6  239.05  9527.5  238.91  9727.3  239.24  9828.6     240
#Mann= 20 ,-1 , 0
 -1503.5     .05       0  -893.5     .08       0  -793.1     .16       0
  1154.2     .12       0  3088.4     .05       0  3208.4     .12       0
  3569.2     .05       0  3944.6     .12       0  4921.4     .07       0
  5058.1     .12       0  5930.6     .05       0    6630     .16       0
    6934     .05       0  7129.6     .16       0  7429.3     .05       0
  7663.3     .16       0  9327.7      .1       0  9427.6     .05       0
  9527.5     .16       0  9727.3     .05       0
#XS Ineff= 2 , 0
       0 3982.09  189.65  6270.9       0     216
Permanent Ineff=
       F       F
Bank Sta=4921.4,5058.1
XS Rating Curve= 0 ,0
Exp/Cntr=0.3,0.1

Type RM Length L Ch R = 1 ,175379  ,1877,1877,1877
BEGIN DESCRIPTION:
NAVASOTA RIVER 277
END DESCRIPTION:
XS GIS Cut Line= 3
      3614814.59     10190946.82      3610124.42     10191212.69
      3604690.92     10191207.24
#Sta/Elev= 30
   302.3  256.22   477.9  245.77   659.2  217.24   814.1  217.12  1008.4  226.94
  1241.4  212.81  1316.4  216.63  1466.5  208.04  1694.7  192.78  2157.8     183
  2812.6  187.84    3550  183.26  4932.2  190.08  4962.2   180.9  5012.1  179.33
  5082.3  188.97  6439.6  187.74  6612.3  192.72  6795.7  211.27  6982.7  214.85
  7289.2   208.4  7387.9  208.52  7486.6  213.88  7585.3  216.94    8700  215.99
  9040.5  221.62  9442.3  238.05 10052.9  239.69 10250.4  239.76 10433.5  238.29
#Mann= 20 ,-1 , 0
   302.3     .05       0   659.2     .16       0   814.1     .16       0
  1241.4     .05       0  1466.5     .16       0  1694.7     .12       0
  2812.6     .12       0  4932.2     .07       0  5082.3     .12       0
  6439.6     .16       0  6795.7      .1       0  6982.7      .1       0
  7289.2     .05       0  7387.9     .12       0  7486.6     .16       0
  7585.3     .05       0    8700     .16       0  9040.5     .05       0
 10052.9      .1       0 10250.4     .05       0
#XS Ineff= 2 , 0
       0 3612.09   187.8  6892.3       0  215.46
Permanent Ineff=
       F       F
Bank Sta=4932.2,5082.3
XS Rating Curve= 0 ,0
Exp/Cntr=0.3,0.1

Type RM Length L Ch R = 1 ,173502  ,1256,1256,1256
BEGIN DESCRIPTION:
NAVASOTA RIVER 278
END DESCRIPTION:
XS GIS Cut Line= 3
      3614269.42     10189812.28      3609935.24     10189576.27
      3604539.01     10190089.62
#Sta/Elev= 30
   659.4  250.27   746.8  252.94  1227.6  234.16  1297.7  236.19  1500.8  222.33
  1659.7   199.9  1798.4  186.93  1988.7  181.34    2229  186.74  2709.7  186.14
  2779.9  180.88  2799.9  186.11  4953.1  189.25  4983.1  179.83  5005.8   179.3
  5033.3  180.84  5053.4  188.93  5892.8  187.79  6020.7  188.17  6320.2  189.75
  6356.1  189.99  6610.4  197.28  6771.1  196.11    6904   206.3  6951.9  210.93
  7334.1  217.27  8800.2  211.71  9091.5  229.41  9834.9  227.88 10420.6  239.89
#Mann= 10 ,-1 , 0
   659.4     .16       0  1659.7     .12       0  4953.1     .07       0
  5053.4     .12       0  5892.8     .05       0  6020.7     .12       0
  6320.2     .05       0  6356.1     .16       0    6904     .05       0
  7334.1     .16       0
#XS Ineff= 2 , 0
         3664.12  188.03
Permanent Ineff=
       F       F
Bank Sta=4953.1,5053.4
XS Rating Curve= 0 ,0
Exp/Cntr=0.3,0.1

Type RM Length L Ch R = 1 ,172246  ,2377,2377,2377
BEGIN DESCRIPTION:
NAVASOTA RIVER 279
END DESCRIPTION:
XS GIS Cut Line= 4
      3614305.32     10189330.64      3611201.12     10188247.29
      3609794.62     10188362.21      3604685.75     10189456.29
#Sta/Elev= 30
     301  231.53   466.7  231.57     575  228.44    1160  212.75  1259.2  202.79
  1480.1  186.18  2743.4  186.98  3026.4  181.19  3111.2  186.89  4929.5  189.85
  4998.5  179.09  5053.7  188.51  5176.4  182.37  6091.1  187.07  6155.8  187.33
  6192.9  188.97  6450.6  199.93  6460.1  199.93  7000.6   198.7  7067.3  198.83
  7360.5  201.46    7548  214.98  7794.7  214.31  8025.4  214.25  8432.6  213.11
  8534.4  210.41  8636.2  210.75  9134.2  230.96  9800.3   225.8 10224.7  231.74
#Mann= 18 ,-1 , 0
     301     .16       0   466.7     .05       0     575     .16       0
  1259.2     .12       0  4929.5     .07       0  5053.7     .12       0
  6091.1     .05       0  6155.8     .12       0  6192.9     .16       0
  6450.6     .05       0  6460.1     .16       0  7000.6     .05       0
  7067.3     .16       0  7794.7     .05       0  8025.4     .16       0
  8432.6     .12       0  8534.4     .07       0  8636.2     .05       0
#XS Ineff= 2 , 0
         3719.53  188.37
Permanent Ineff=
       F       F
Bank Sta=4929.5,5053.7
XS Rating Curve= 0 ,0
Exp/Cntr=0.3,0.1

Type RM Length L Ch R = 1 ,169869  ,2422,2422,2422
BEGIN DESCRIPTION:
NAVASOTA RIVER 069
END DESCRIPTION:
XS GIS Cut Line= 3
      3615859.01     10186513.18      3607213.23     10186325.68
      3605109.09     10188971.48
#Sta/Elev= 30
   -1431  235.76 -1129.2   233.2    -884  208.41  -631.3  196.52      -4  184.36
   176.3   179.4   286.3  186.09  1700.5  184.31    1885  184.62  4917.4  188.05
  4947.4  179.49  5007.2  178.87  5037.4  179.75  5057.4  188.19  5076.8  188.84
  5208.2  188.22  5352.9  187.43  5374.2  187.36  5710.8  186.22  6009.1  187.24
  6337.7  188.25  6877.9   206.3  7461.2  206.29    7873  207.87    8199  210.66
  8644.7  208.47  8936.5  215.48  9570.6  208.26    9891  219.85 10597.3  224.72
#Mann= 16 ,-1 , 0
   -1431     .16       0  -631.3     .05       0      -4     .12       0
  1700.5     .07       0    1885     .12       0  4917.4     .07       0
  5057.4     .16       0  5076.8     .12       0  5208.2     .16       0
  5352.9     .05       0  5374.2     .16       0  5710.8     .12       0
  6009.1     .16       0  7461.2     .05       0    7873     .16       0
    8199     .05       0
#XS Ineff= 2 , 0
         2300.71  185.69
Permanent Ineff=
       F       F
Bank Sta=4917.4,5057.4
XS Rating Curve= 0 ,0
Exp/Cntr=0.3,0.1

Type RM Length L Ch R = 1 ,167447  ,1542,1542,1542
BEGIN DESCRIPTION:
NAVASOTA RIVER 280
END DESCRIPTION:
XS GIS Cut Line= 3
      3616270.24     10185963.96      3609869.75     10184307.77
      3603235.59     10183586.07
#Sta/Elev= 30
 -1611.3  245.75 -1300.4  239.71 -1021.2  216.63  -654.9  200.33  -376.8  199.57
   -44.4  196.04      50   191.9   123.3  181.35   232.7  179.06   235.5  178.56
   238.7  179.06   514.6  186.07  1968.8  184.46  2035.4  184.44  4242.4  185.66
  4478.5  186.67  4683.8  181.41  4800.5  188.08  4935.6  187.33    4963  179.49
  5027.8  179.29  5088.2   188.5  6832.1   186.2  6941.9  186.33 10257.4  186.35
 10273.4  186.43 10929.4  186.86 11083.3  198.41 11324.7  226.79 11673.3  234.45
#Mann= 19 ,-1 , 0
 -1611.3     .16       0  -654.9     .05       0  -376.8     .16       0
   -44.4     .12       0      50     .16       0   123.3     .12       0
   232.7     .07       0   238.7     .12       0  1968.8     .07       0
  2035.4     .12       0  4242.4     .07       0  4478.5     .12       0
  4800.5     .07       0  5088.2     .12       0  6832.1     .07       0
  6941.9     .12       0 10257.4     .07       0 10273.4     .12       0
 10929.4     .16       0
#XS Ineff= 2 , 0
          515.32   186.1
Permanent Ineff=
       F       F
Bank Sta=4800.5,5088.2
XS Rating Curve= 0 ,0
Exp/Cntr=0.3,0.1

Type RM Length L Ch R = 1 ,165905  ,3938,3938,3938
BEGIN DESCRIPTION:
NAVASOTA RIVER 281
END DESCRIPTION:
XS GIS Cut Line= 3
      3616446.08     10185677.07      3609762.09     10182833.81
       3602946.6     10183076.35
#Sta/Elev= 30
 -2263.6  241.81 -2034.5  239.92 -1547.3  201.37 -1261.5  201.66    -717  198.37
  -531.4  201.62  -364.8  188.65  -227.1  179.11   401.1  184.02   806.3   179.4
  1152.8  184.91  1468.5  184.75  2242.1  183.47  2745.1  184.45  3069.4  184.83
  3384.4   185.2    3755  185.57  4804.4  188.06    4997  178.55    5050  188.04
  5420.2  179.65  6351.4   184.8  6552.6  185.54  9942.6  185.35 10312.4  185.71
 11001.3  186.07   11314  212.86   11414  205.94 11514.1  223.77 11819.8  235.41
#Mann= 20 ,-1 , 0
 -2263.6     .16       0 -1261.5     .05       0    -717     .16       0
  -364.8     .12       0   401.1     .12       0   806.3     .12       0
  1152.8     .07       0  1468.5     .12       0  2242.1     .12       0
  2745.1     .12       0  3069.4     .12       0  3384.4     .07       0
    3755     .12       0  4804.4     .07       0    5050     .12       0
  6351.4     .07       0  6552.6     .12       0  9942.6     .07       0
 10312.4     .12       0 11001.3     .16       0
#XS Ineff= 2 , 0
          859.73  185.49 5518.79          188.42
Permanent Ineff=
       F       F
Bank Sta=4804.4,5050
XS Rating Curve= 0 ,0
Exp/Cntr=0.3,0.1

Type RM Length L Ch R = 1 ,161967  ,3112,3112,3112
BEGIN DESCRIPTION:
NAVASOTA RIVER 282
END DESCRIPTION:
XS GIS Cut Line= 3
      3617095.69     10185185.19      3611050.94     10181455.09
       3602340.9     10181487.13
#Sta/Elev= 30
   -2103  224.75 -1933.6  218.85   -1534  206.16  -190.4  196.36   445.6  203.28
   586.6  196.92   784.7  188.57  3200.8  183.39  3316.6  177.71  3380.7  183.59
  4805.7  186.24  4951.6  184.96  4986.9  178.34  5048.8  186.26  6086.5  187.32
  6647.2  185.62  7349.4  181.12  7526.6  185.31  7898.9  180.44  7928.9  186.07
  8901.3  185.45  9131.1  185.08 10088.3  184.72 10487.2  184.57 12378.9  183.99
 12670.6  191.94 13128.9  231.37 13218.6  230.99 13460.4  227.96 13710.1  234.15
#Mann= 19 ,-1 , 0
   -2103     .05       0 -1933.6     .05       0   -1534     .16       0
  -190.4     .05       0   586.6     .16       0   784.7     .12       0
  4805.7     .07       0  5048.8     .12       0  6086.5     .16       0
  6647.2     .12       0  7349.4     .07       0  7526.6     .12       0
  8901.3     .07       0  9131.1     .12       0 10088.3     .07       0
 10487.2     .12       0 12670.6     .05       0 13218.6     .16       0
 13460.4     .05       0
#XS Ineff= 2 , 0
          445.64  203.26 6009.03          188.74
Permanent Ineff=
       F       F
Bank Sta=4805.7,5048.8
XS Rating Curve= 0 ,0
Exp/Cntr=0.3,0.1

Type RM Length L Ch R = 1 ,158855  ,1146,1146,1146
BEGIN DESCRIPTION:
NAVASOTA RIVER 283
END DESCRIPTION:
XS GIS Cut Line= 5
       3617201.2     10184739.26      3614032.42     10181816.49
      3612925.84     10181245.06      3612096.65     10180852.95
      3602937.91     10180207.18
#Sta/Elev= 30
  -556.3  220.84    -478  219.42     354  200.39  1558.1  195.68  1906.5  197.62
  1946.9  197.61  2206.1  197.53  2209.2  197.53  2335.7  197.49  2508.4  197.43
  2880.8  196.43  2909.2  200.62  2958.5  195.28  3184.8  190.08  3397.4   187.1
  3562.5  190.14  4344.3  181.89  4857.9  183.96  4958.9  177.54  5258.8  184.94
    6783  184.27  6940.1     185  6964.4  182.23  6977.1  184.78  7232.1  185.91
 11395.3  181.73 13315.1  185.59 13318.3  185.59 14450.7  188.48 15098.7  234.97
#Mann= 19 ,-1 , 0
  -556.3     .05       0    -478     .16       0  1558.1     .05       0
  1906.5     .08       0  1946.9     .05       0  2206.1     .08       0
  2209.2     .05       0  2335.7     .08       0  2508.4     .05       0
  3562.5     .12       0  4857.9     .07       0  5258.8     .12       0
    6783     .07       0  6940.1     .12       0  6977.1     .07       0
  7232.1     .12       0 13315.1     .07       0 13318.3     .12       0
 14450.7     .16       0
#XS Ineff= 2 , 0
         2906.58  200.66 5925.66          185.64
Permanent Ineff=
       F       F
Bank Sta=4857.9,5258.8
XS Rating Curve= 0 ,0
Exp/Cntr=0.3,0.1

Type RM Length L Ch R = 1 ,157709  ,2196,2196,2196
BEGIN DESCRIPTION:
NAVASOTA RIVER 284
END DESCRIPTION:
XS GIS Cut Line= 3
      3618216.63     10180832.88      3613903.62     10180705.47
      3602912.72     10180164.47
#Sta/Elev= 30
   685.1   224.3  1007.2  199.61  1159.8  194.03  1419.9  194.95    1460  189.17
  1569.4  199.12  1771.5  198.93  2370.4  195.56  2500.4  199.63  3254.7  192.69
  3353.3  188.12  3510.6  185.68  3772.4  184.08  3912.8  185.05    4168  185.61
  4321.3   185.5  4480.5  185.38  4661.4  179.93  4941.5  184.56  4971.2  177.94
  5151.7  185.34  7443.7  184.42  7707.4  185.22  8301.8  185.04  8310.2  185.04
 14057.9  184.12 14166.6  184.66 15083.7  183.42 15307.4  189.62 16004.2  236.82
#Mann= 20 ,-1 , 0
   685.1     .05       0  1007.2     .12       0  1771.5     .16       0
  3254.7     .08       0  3353.3     .05       0  3510.6     .12       0
  3772.4     .05       0  3912.8     .05       0    4168     .12       0
  4321.3     .05       0  4480.5     .12       0  4941.5     .07       0
  5151.7     .12       0  7443.7     .07       0  7707.4     .12       0
  8301.8     .07       0  8310.2     .12       0 14057.9     .07       0
 14166.6     .12       0 15307.4     .16       0
#XS Ineff= 2 , 0
         2502.53  199.54 6085.46          185.68
Permanent Ineff=
       F       F
Bank Sta=4941.5,5151.7
XS Rating Curve= 0 ,0
Exp/Cntr=0.3,0.1

Type RM Length L Ch R = 1 ,155513  ,4674,4674,4674
BEGIN DESCRIPTION:
NAVASOTA RIVER 285
END DESCRIPTION:
XS GIS Cut Line= 3
      3618866.25     10179667.98       3613737.3     10179191.93
      3601660.52     10179138.04
#Sta/Elev= 30
    -151  223.19   359.7  215.11     656  209.93  1388.9  189.64  2027.5  186.58
  2062.6  196.74  2156.6  197.22  2956.4  197.08  3368.1  185.71    3833  185.63
  4211.7  185.23  4754.1  184.66  4949.5  183.32  5004.9  176.55  5055.2  184.73
  5235.2  185.04  6104.5  183.27  6279.2  183.69  7033.1  182.93  7368.7   183.2
 10960.8  184.51 11091.9  184.61 11317.8  184.72 14885.3  181.63 15212.8  186.42
   15574  187.68 16095.3  190.01 16290.9  198.89 16655.3   231.8 17076.9  237.38
#Mann= 20 ,-1 , 0
    -151     .05       0   359.7     .08       0     656     .05       0
  1388.9     .12       0  2156.6     .16       0  3368.1     .05       0
    3833     .05       0  4211.7     .12       0  4754.1     .07       0
  5235.2     .12       0  6104.5     .07       0  6279.2     .12       0
  7033.1     .12       0  7368.7     .12       0 10960.8     .16       0
 11091.9     .12       0 11317.8     .12       0 15212.8     .05       0
   15574     .12       0 16290.9     .05       0
#XS Ineff= 2 , 0
          2787.6  198.17
Permanent Ineff=
       F       F
Bank Sta=4754.1,5235.2
XS Rating Curve= 0 ,0
Exp/Cntr=0.3,0.1

Type RM Length L Ch R = 1 ,150839  ,1073,1073,1073
BEGIN DESCRIPTION:
NAVASOTA RIVER 210
END DESCRIPTION:
XS GIS Cut Line= 4
      3618648.14     10179263.77       3613405.9      10177086.5
      3605909.46     10173972.99        3602090.      10170570.2
#Sta/Elev= 30
  -676.4  219.98  -212.1  199.89   100.8  205.73   845.3   207.7  1128.1   197.1
    1538  184.08  2773.1   182.5  4939.1  182.72  4969.6  175.62  5058.3  182.29
  5312.6  182.49  7505.5  182.97  8441.9  182.69 12094.8  182.03 13146.9  183.34
 15372.7  184.21 15943.6  184.43 16254.1  184.55 16423.8  188.58 16519.4     198
 16700.5  218.23 17082.3  221.79 17139.5  216.67 17479.4  230.31 17592.7  230.08
   17642  222.63 17711.7  226.84 17918.7  215.14   18052  225.63 18232.7   228.7
#Mann= 20 ,-1 , 0
  -676.4     .05       0   100.8     .05       0   845.3     .16       0
  1128.1     .05       0    1538     .07       0  2773.1     .12       0
  4939.1     .07       0  5058.3     .12       0  5312.6     .12       0
  7505.5     .16       0  8441.9     .12       0 12094.8     .12       0
 13146.9     .12       0 15372.7     .12       0 15943.6     .12       0
 16519.4     .05       0 17082.3     .16       0 17479.4     .05       0
 17711.7     .16       0   18052     .05       0
#XS Ineff= 2 , 0
           829.7  208.2416990.13          224.36
Permanent Ineff=
       F       F
Bank Sta=4939.1,5058.3
XS Rating Curve= 0 ,0
Exp/Cntr=0.3,0.1

Type RM Length L Ch R = 1 ,149766  ,1448,1448,1448
BEGIN DESCRIPTION:
NAVASOTA RIVER 211
END DESCRIPTION:
XS GIS Cut Line= 5
       3618725.5     10179214.81      3617487.62     10178001.23
      3614138.16     10176363.11      3611274.76     10175124.43
      3608652.52     10170292.45
#Sta/Elev= 30
  -462.1  221.34  -396.4  220.74   108.2   194.7   334.8  190.94  1593.1  182.06
    1935  182.13  2235.5  182.19  3105.9  182.37  4007.7  182.56    4929  183.48
  4990.8  175.71    5072  183.13  5764.9  182.04  6975.5  182.25  7338.7  182.13
  7650.2  182.02 10165.5  181.42 10674.3  181.31 11174.6  182.83 11873.9     186
 12415.5  189.39 12459.2  194.71 12526.2  218.97   12617  213.71 12799.2  232.29
 12838.9  242.17 13146.4  235.91   13425  257.49 13571.5  253.97 13617.5  255.28
#Mann= 20 ,-1 , 0
  -462.1     .08       0  -396.4     .05       0   334.8     .05       0
  1593.1     .12       0    1935     .12       0  2235.5     .07       0
  3105.9     .12       0  4007.7     .12       0    4929     .07       0
    5072     .12       0  5764.9     .12       0  6975.5     .12       0
  7338.7     .16       0  7650.2     .12       0 10165.5     .05       0
 10674.3     .12       0 11174.6     .12       0 11873.9     .16       0
 12838.9     .05       0 13571.5     .16       0
#XS Ineff= 2 , 0
                        12881.78          246.15
Permanent Ineff=
       F       F
Bank Sta=4929,5072
XS Rating Curve= 0 ,0
Exp/Cntr=0.3,0.1

Type RM Length L Ch R = 1 ,148318  ,1711,1711,1711
BEGIN DESCRIPTION:
NAVASOTA RIVER 364
END DESCRIPTION:
XS GIS Cut Line= 4
      3619260.55      10179396.1      3617524.42     10177464.66
      3612055.29     10173313.27       3610736.5     10170363.33
#Sta/Elev= 30
  -666.8  222.89  -501.6  213.17    71.7  206.51   593.4  188.71   865.1  185.85
  1124.9  183.11  1261.9  181.67  1392.6  181.68  1758.7  182.12  1941.1  182.04
  2581.4  181.72  2944.4   181.8  3468.3  181.92  3904.5  182.02    4331  182.12
  4536.3  182.17  4932.3  181.76  5017.3  175.03  5059.2  183.05    6045   177.1
  9351.3   182.2  9788.3  182.85 10185.5     183 10608.2  193.77 10654.6  197.57
   10701   217.1 10967.1     207 11221.1  227.05 11695.6  244.29 12027.8  245.09
#Mann= 20 ,-1 , 0
  -666.8     .05       0   593.4     .07       0   865.1     .12       0
  1124.9     .07       0  1261.9     .12       0  1392.6     .07       0
  1758.7     .12       0  1941.1     .07       0  2581.4     .07       0
  2944.4     .07       0  3468.3     .12       0  3904.5     .12       0
    4331     .07       0  4536.3     .12       0  4932.3     .07       0
  5059.2     .12       0  9351.3     .05       0  9788.3     .12       0
 10185.5     .16       0 11695.6     .05       0
#XS Ineff= 2 ,-1
  5909.8    6095  182.2110700.84 11117.4  217.06
Permanent Ineff=
       F       F
Bank Sta=4932.3,5059.2
XS Rating Curve= 0 ,0
Exp/Cntr=0.3,0.1

Type RM Length L Ch R = 1 ,146607  ,1330,1330,1330
BEGIN DESCRIPTION:
NAVASOTA RIVER 365
END DESCRIPTION:
XS GIS Cut Line= 4
      3619482.36     10179346.93      3618375.58     10177159.41
      3615198.07     10174321.48      3610949.37     10170467.58
#Sta/Elev= 30
 -1711.9   215.7  -842.3  192.46  -515.2  189.49  -165.5   187.3      29  186.08
     738  181.63  4138.7   182.3  4413.5   181.5  4926.5  181.74  4961.4  174.92
  5075.2  181.29  5669.6  181.71  5711.8  176.82  7856.8  180.84  8384.9  186.59
  8535.1  188.48  8911.7   220.5  9096.2  221.42  9520.6   236.4  9617.5  233.88
  9750.2  233.79  9903.1  233.69 10003.5  233.63   10056   233.6 10132.2  233.78
 10260.9  233.78 10320.8  231.93 10428.1  243.11 10513.4  249.43 10736.2  254.04
#Mann= 20 ,-1 , 0
 -1711.9     .05       0  -842.3     .05       0  -515.2     .07       0
  -165.5     .12       0      29     .07       0  4138.7     .07       0
  4413.5     .12       0  4926.5     .07       0  5075.2     .12       0
  8384.9     .16       0  8535.1     .16       0  9617.5      .1       0
  9750.2     .08       0  9903.1     .08       0 10003.5     .05       0
   10056      .1       0 10132.2     .05       0 10260.9     .05       0
 10428.1     .16       0 10513.4     .05       0
Bank Sta=4926.5,5075.2
XS Rating Curve= 0 ,0
Exp/Cntr=0.3,0.1

Type RM Length L Ch R = 1 ,145277  ,4278,4278,4278
BEGIN DESCRIPTION:
NAVASOTA RIVER 366
END DESCRIPTION:
XS GIS Cut Line= 4
      3619562.91     10179310.49      3618822.45       10176866.
      3616178.28       10173847.      3611020.34     10170436.71
#Sta/Elev= 30
 -1567.4  213.78  -622.8  192.59  -103.2  182.67   267.7  182.09   787.8  181.71
  1278.7  181.53  1715.7  181.49  3082.4  181.36  3505.9  181.32  4073.8  181.27
  4826.9  181.81  4944.2  181.49  5007.1   174.7  5058.2  180.94  6541.1   179.5
  6743.2  180.62  7844.9  180.55    8400  187.29  8693.6  197.52    8826  203.08
  9244.3  198.87  9713.8  242.69 10086.3  246.93 10262.2  243.34 10492.9  234.05
 10622.6   241.5 10654.6  237.76 10797.2  235.02 10998.8  253.37 11183.4  256.42
#Mann= 20 ,-1 , 0
 -1567.4     .05       0  -622.8     .05       0  -103.2     .12       0
   267.7     .07       0   787.8     .12       0  1278.7     .12       0
  1715.7     .07       0  3082.4     .12       0  3505.9     .12       0
  4073.8     .12       0  4826.9     .12       0  4944.2     .07       0
  5058.2     .12       0  6541.1     .07       0  6743.2     .12       0
  8693.6     .16       0 10086.3     .16       0 10262.2     .05       0
 10492.9     .08       0 10654.6     .05       0
Bank Sta=4944.2,5058.2
XS Rating Curve= 0 ,0
Exp/Cntr=0.3,0.1

Type RM Length L Ch R = 1 ,140999  ,1321,1321,1321
BEGIN DESCRIPTION:
NAVASOTA RIVER 367
END DESCRIPTION:
XS GIS Cut Line= 4
      3622734.77     10175211.03      3616537.72     10171858.42
      3615384.09     10171544.85      3611102.78     10170319.52
#Sta/Elev= 30
 -3241.3  221.76 -2770.4   212.1 -2296.7  209.22 -2076.9  210.03 -1757.8  209.83
 -1669.3  200.06   -1108  187.23   124.3  184.69   230.8  184.65   450.6  183.85
   650.2  183.08   863.1  182.27    1015  181.75  1286.3   181.1  1723.7  180.66
  1890.4  180.76  3221.5   181.6  3416.2  181.72  4289.1  179.96  4418.9  181.47
  4989.6  173.25  5101.7  180.77  7199.5  184.91  7323.1  190.71  7385.6  207.24
  7415.2  217.42  8229.9  218.59  8341.6  229.88  8507.4   221.9  9453.2  250.59
#Mann= 20 ,-1 , 0
 -3241.3     .05       0 -2770.4     .05       0 -2296.7     .08       0
 -2076.9     .05       0   124.3     .05       0   230.8      .1       0
   450.6     .16       0   650.2     .12       0   863.1     .12       0
    1015     .05       0  1286.3     .12       0  1723.7     .07       0
  1890.4     .05       0  3221.5     .12       0  3416.2     .05       0
  4289.1     .12       0  4418.9     .07       0  5101.7     .12       0
  7199.5     .16       0  7385.6     .05       0
Bank Sta=4418.9,5101.7
XS Rating Curve= 0 ,0
Exp/Cntr=0.3,0.1

Type RM Length L Ch R = 1 ,139678  ,2361,2361,2361
BEGIN DESCRIPTION:
NAVASOTA RIVER 417
END DESCRIPTION:
XS GIS Cut Line= 3
        3622814.     10175135.15      3616112.94       10170680.
      3612332.27      10169797.5
#Sta/Elev= 30
 -3046.9  220.25 -2271.5  201.32   -2192  202.01   -2156  207.66 -1849.2  209.96
 -1733.6  208.78 -1667.8  207.12 -1477.9  197.77   -1060  186.34   754.1  181.56
    1250  181.52  2670.7  185.43  2697.8  182.25  3268.9  182.38  3434.3  178.06
  3720.1  181.43  4495.5  176.65  4847.2  181.41  5021.1  173.39  5063.2  179.67
  5206.2  180.79  5247.3  177.56  5674.1  181.43  7730.9  180.97  7962.8   184.1
  8081.5   192.8  8265.7  214.06    8482  215.86  8687.4   230.4  8882.3  232.85
#Mann= 10 ,-1 , 0
 -3046.9     .05       0 -1849.2     .08       0 -1733.6      .1       0
 -1667.8     .05       0   754.1     .12       0    1250     .05       0
  3720.1     .12       0  4847.2     .07       0  5206.2     .12       0
  7730.9     .16       0
#XS Ineff= 2 ,-1
 -2719.4 -1867.8  210.05 -1867.8  2661.7  185.35
Permanent Ineff=
       F       F
Bank Sta=4847.2,5206.2
XS Rating Curve= 0 ,0
Exp/Cntr=0.3,0.1

Type RM Length L Ch R = 1 ,137317  ,1078,1078,1078
BEGIN DESCRIPTION:
NAVASOTA RIVER 418
END DESCRIPTION:
XS GIS Cut Line= 5
      3624656.23     10175268.83      3621723.04     10172891.21
      3617817.62     10170590.94      3616661.35     10169991.21
        3612328.     10169713.43
#Sta/Elev= 30
 -3308.3   226.9 -3172.6  223.94 -2447.1  193.02 -1186.5   182.9   -1081  185.82
 -1022.5  185.68  -957.9  185.53  -711.6  184.95   417.4  186.06  1298.8  180.31
  1410.8  184.25  3146.8     183  3202.2  182.99  3354.2  182.95  3431.4  182.93
  4881.6  178.53  4936.8   181.3  4967.4  174.54  5010.3  173.34  5165.5  180.44
    5761  181.27  5884.9  175.29    5930  178.73    6392   179.9  6432.1  175.14
  6790.6  179.18  7057.5  179.76    9812  185.74 10099.6  207.72 10644.8  230.87
#Mann= 19 ,-1 , 0
 -3308.3     .16       0 -3172.6     .05       0 -1186.5     .12       0
   -1081     .07       0 -1022.5     .05       0  -957.9     .07       0
  -711.6     .05       0  1298.8     .07       0  1410.8     .05       0
  3146.8     .12       0  3202.2     .08       0  3354.2     .12       0
  3431.4     .05       0  4881.6     .07       0  4936.8    .033       0
  5165.5     .12       0  6790.6     .07       0  7057.5     .12       0
    9812     .16       0
#XS Ineff= 2 , 0
       0  1396.9  184.58               0
Permanent Ineff=
       F       F
Bank Sta=4936.8,5165.5
XS Rating Curve= 0 ,0
Exp/Cntr=0.3,0.1

Type RM Length L Ch R = 1 ,136239  ,1829,1829,1829
BEGIN DESCRIPTION:
NAVASOTA RIVER 141
END DESCRIPTION:
XS GIS Cut Line= 3
      3625492.78     10168725.59      3621846.96     10169611.01
      3612237.59     10169637.05
#Sta/Elev= 30
 -2908.4  225.94 -2501.7  215.49 -2399.1  212.53 -2099.4  192.14 -1801.9  183.76
  -930.2  183.73  -376.2  186.78  1278.3  183.06  1318.3  179.41  1388.3  183.76
  1551.6   182.9  1904.7  182.17  3170.2  181.46  3940.7  181.29  4132.3  181.17
  4434.3  177.62  4597.4  178.66  4938.3   180.7    4988  173.33  5068.3  179.34
  5218.3  181.23  5520.1  181.21  5717.5  181.19  5945.5  181.17  6104.5  181.16
  6842.4  180.83  8778.3  179.96  9533.8  186.05 10308.3   227.6 10452.8  227.37
#Mann= 19 ,-1 , 0
 -2908.4     .05       0 -2501.7     .08       0 -2399.1     .05       0
  -930.2     .12       0  1551.6     .05       0  1904.7     .12       0
  3170.2     .05       0  3940.7     .12       0  4132.3     .05       0
  4434.3     .12       0  4597.4     .12       0  4938.3     .07       0
  5218.3     .07       0  5520.1     .12       0  5717.5     .12       0
  5945.5     .07       0  6104.5     .12       0  6842.4     .12       0
  9533.8     .16       0
#XS Ineff= 2 , 0
         -375.94   186.8
Permanent Ineff=
       F       F
Bank Sta=4938.3,5218.3
XS Rating Curve= 0 ,0
Exp/Cntr=0.3,0.1

Type RM Length L Ch R = 1 ,134410  ,3283,3283,3283
BEGIN DESCRIPTION:
NAVASOTA RIVER 474
END DESCRIPTION:
XS GIS Cut Line= 3
      3622738.23      10167750.1      3618157.21      10168302.4
      3609905.55     10169425.25
#Sta/Elev= 30
   385.8   231.4   684.1  218.65   734.4  206.58   959.6  196.28  1002.1  194.71
  1502.3  188.31  1761.8  195.25  2102.5  182.99  3272.7  180.54    3313  174.34
  3428.2  180.58  3680.1  181.41  4934.6  180.13    5015  173.03  5136.3  179.86
  5376.2   177.3  5526.4  177.54  9961.5  183.74 10071.7  184.73 10138.2  187.06
 10664.9  196.28 10777.9  190.28 10828.3  197.41 11114.5  207.92 11414.2  208.33
 11443.9  202.72 11502.3  208.73 11567.6  210.83 11751.9  216.48 13327.7  230.74
#Mann= 17 ,-1 , 0
   385.8     .05       0   959.6     .16       0  1002.1     .05       0
  1502.3     .16       0  2102.5     .12       0  3428.2     .07       0
  3680.1     .12       0  4934.6     .07       0  5136.3     .12       0
  5376.2     .07       0  5526.4     .12       0  9961.5     .16       0
 10071.7     .12       0 10138.2     .16       0 11502.3     .05       0
 11567.6     .16       0 11751.9     .05       0
#XS Ineff= 2 , 0
         1762.24  195.23
Permanent Ineff=
       F       F
Bank Sta=4934.6,5136.3
XS Rating Curve= 0 ,0
Exp/Cntr=0.3,0.1

Type RM Length L Ch R = 1 ,131127  ,1795,1795,1795
BEGIN DESCRIPTION:
NAVASOTA RIVER 427
END DESCRIPTION:
XS GIS Cut Line= 3
      3621477.75      10166430.5      3619296.27     10166793.02
       3609795.4      10169268.6
#Sta/Elev= 30
  2788.6  237.15  2883.8  238.26  2936.2  228.39  3220.1  208.25    3498  204.75
  3675.6  184.58  4199.3  179.21  4397.5  177.84    4904  179.38  4993.8  172.27
  5035.3  179.35  5758.7  179.51  5806.4  175.05  6241.5  180.49  7145.4  179.99
  7328.7  180.24    7661     180  8131.9  179.73  8444.2  180.08  8642.4  180.13
  8861.8  180.04  9084.7  180.65 10763.9   182.1 11352.4  186.42 11805.7  193.16
 12062.6  207.45 12713.5  207.86 13753.7  219.01   14280  225.12 14818.1  230.41
#Mann= 20 ,-1 , 0
  2788.6     .05       0  4199.3     .07       0  4397.5     .12       0
    4904     .07       0  5035.3     .12       0  7145.4     .12       0
  7328.7     .07       0    7661     .12       0  8131.9     .12       0
  8444.2     .07       0  8642.4     .12       0  8861.8     .07       0
  9084.7     .12       0 10763.9     .05       0 11352.4     .16       0
 11805.7     .05       0 12062.6     .16       0 12713.5     .05       0
 13753.7     .16       0   14280     .05       0
Bank Sta=4904,5035.3
XS Rating Curve= 0 ,0
Exp/Cntr=0.3,0.1

Type RM Length L Ch R = 1 ,129332  ,1425,1425,1425
BEGIN DESCRIPTION:
NAVASOTA RIVER 426
END DESCRIPTION:
XS GIS Cut Line= 3
      3621830.31     10165047.04      3619295.75     10165094.06
      3609429.08     10168704.82
#Sta/Elev= 30
    2465  229.97  2980.5  216.61  3513.4  208.41  3883.5  207.46  4143.5  191.83
  4501.3  180.56  4643.6  177.28  4943.6  178.38  5014.3  171.64  5057.1  178.82
    7618  181.99  7916.8  190.55  8016.5  196.44  8151.8  202.07  8451.2  202.37
    9061  197.87  9166.6   199.7  9515.6  205.03  9891.1  201.95   10818  204.42
 11231.2  190.21 11850.9  197.22   12362  197.99 12743.8  205.03 13583.6     210
 14370.8  215.63 14427.9  212.83 15101.6  223.13 15208.2   224.1 15506.6  227.51
#Mann= 13 ,-1 , 0
    2465     .05       0  4501.3     .12       0  4943.6     .07       0
  5057.1     .12       0    7618     .05       0  8016.5     .16       0
  8151.8     .05       0  8451.2     .16       0  9166.6     .05       0
 13583.6     .16       0 14370.8     .05       0 15101.6      .1       0
 15208.2     .16       0
Bank Sta=4943.6,5057.1
XS Rating Curve= 0 ,0
Exp/Cntr=0.3,0.1

Type RM Length L Ch R = 1 ,127907  ,1687,1687,1687
BEGIN DESCRIPTION:
NAVASOTA RIVER 425
END DESCRIPTION:
XS GIS Cut Line= 3
      3622839.93     10164161.62        3618427.     10164360.21
      3609443.19     10168263.19
#Sta/Elev= 30
   582.6  231.77    1171   203.2  1461.3  202.45  1501.4  196.92  1841.7  202.98
  2470.6  190.27  3393.3  190.72  3503.4  185.77  4370.8  181.32  4611.6  180.09
  4661.7  179.83  4874.8  179.55  5018.7  171.44  5059.8  179.61  6279.4  177.99
  6354.5  177.24  7972.3   183.3    8418   203.7  9009.3   203.2  9050.3   195.3
  9236.7  204.69  9983.9  202.81 10310.5  193.95   10917  191.78 12019.7  200.38
 12288.5  197.18 12830.8  206.36 13667.6  215.38 14120.2  216.55   14795  229.57
#Mann= 11 ,-1 , 0
   582.6     .05       0  4370.8     .12       0  4611.6     .05       0
  4661.7     .12       0  4874.8     .07       0  5059.8     .12       0
  6279.4     .07       0  6354.5     .12       0  7972.3     .05       0
 12830.8     .16       0 13667.6     .05       0
Bank Sta=4874.8,5059.8
XS Rating Curve= 0 ,0
Exp/Cntr=0.3,0.1

Type RM Length L Ch R = 1 ,126220  ,4177,4177,4177
BEGIN DESCRIPTION:
NAVASOTA RIVER 424
END DESCRIPTION:
XS GIS Cut Line= 3
      3623073.37     10162898.17      3618618.66      10163117.5
       3615521.3     10162984.97
#Sta/Elev= 30
   539.9  221.75   553.8  222.22   781.5   222.3   821.5  213.33   871.6  207.19
  1041.8  194.89  1782.7  184.67    2874  181.44  3424.7  186.28    3735  184.07
  4445.9  187.88    4672  182.46  4826.3     178  4956.5  178.56  4976.5  175.36
  4981.8   170.9  5136.7  178.14  5766.4  179.03  5915.4  176.78  5967.4  172.61
  5997.5  177.39  6070.8  178.51  6461.7  175.88  7097.4  180.04  7196.2  180.33
  7270.6  180.82  7498.8   187.9  7671.8  206.09  7969.3  235.87  8100.2  240.15
#Mann= 13 ,-1 , 0
   539.9      .1       0   553.8     .05       0    4672     .12       0
  4956.5     .07       0  5136.7     .12       0  5766.4     .07       0
  5915.4     .12       0  6070.8     .07       0  6461.7     .12       0
  7097.4     .05       0  7196.2     .12       0  7270.6     .05       0
  7671.8     .16       0
Bank Sta=4956.5,5136.7
XS Rating Curve= 0 ,0
Exp/Cntr=0.3,0.1

Type RM Length L Ch R = 1 ,122043  ,1522,1522,1522
BEGIN DESCRIPTION:
NAVASOTA RIVER 249
END DESCRIPTION:
XS GIS Cut Line= 3
      3623155.26     10161006.03      3620475.09     10161266.45
      3615190.83     10160615.41
#Sta/Elev= 30
  -632.1  220.89  -367.7  208.01  -136.6  216.65   114.6  199.81   625.4  186.16
  1110.4   182.5  1579.6  182.56  1679.1     183  1878.2  184.33  2658.2  197.37
  3066.8  187.24  3357.8  184.56    4133  180.41  4392.9  178.89  4925.8  177.77
  5001.7  168.53  5126.7  178.61  5596.1  178.85  5918.2  177.06  6035.7  178.34
  6240.2  184.09  6355.9  193.11  6446.6  224.03  6486.9  227.71  6859.7  208.09
    7023   215.5  7133.1  225.79    7172  240.97  7322.2  243.23  7384.9  243.56
#Mann= 18 ,-1 , 0
  -632.1     .16       0   625.4     .12       0  1110.4     .12       0
  1579.6     .16       0  1679.1     .05       0  1878.2     .16       0
  3066.8     .05       0  3357.8     .05       0    4133     .12       0
  4392.9     .12       0  4925.8     .07       0  5126.7     .12       0
  5596.1     .07       0  5918.2     .12       0  6035.7     .05       0
  6240.2     .16       0    7023     .05       0  7322.2     .08       0
Bank Sta=4925.8,5126.7
XS Rating Curve= 0 ,0
Exp/Cntr=0.3,0.1

Type RM Length L Ch R = 1 ,120521  ,1526,1526,1526
BEGIN DESCRIPTION:
NAVASOTA RIVER 423
END DESCRIPTION:
XS GIS Cut Line= 3
      3623053.91     10160549.65      3617953.56     10159943.02
      3617049.99     10159396.87
#Sta/Elev= 30
  -136.3  227.12   348.9  219.86   530.2  204.06   646.5  200.12   701.4   195.4
   852.4  202.01  1134.4  201.07  1386.2     194    1930     201    2437  196.69
    2488  195.06  2890.6  186.98  2977.3  189.77  3228.4  181.94  3327.3  179.49
  3667.1  179.39    3686  179.46  4920.9  177.17  4961.2  169.62    5031  168.34
    5074   176.6  5231.7  177.04    5301  184.62    5365  211.55  5544.9  217.47
  5687.1  210.88  5760.8  227.86  5836.8  231.88  5878.7  232.49  6055.8  231.33
#Mann= 15 ,-1 , 0
  -136.3     .16       0   646.5     .05       0    2437     .16       0
    2488     .05       0  2890.6     .16       0  3228.4     .05       0
  3327.3     .12       0  3667.1     .16       0    3686     .12       0
  4920.9     .07       0    5074     .12       0  5231.7     .16       0
  5544.9     .05       0  5836.8      .1       0  5878.7     .05       0
Bank Sta=4920.9,5074
XS Rating Curve= 0 ,0
Exp/Cntr=0.3,0.1

Type RM Length L Ch R = 1 ,118995  ,3173,3173,3173
BEGIN DESCRIPTION:
NAVASOTA RIVER 422
END DESCRIPTION:
XS GIS Cut Line= 3
      3621896.44      10159369.8      3618511.89     10158743.54
      3616346.31     10158487.23
#Sta/Elev= 30
    1558  227.11  1687.4  223.16  1969.2  207.24    2126  191.07    2254  183.02
  2499.2  178.89  4043.7  178.96  4159.7  173.31  4212.6  177.06  4318.4  178.53
  4420.1  175.19  4540.2  175.43  4633.7  178.97  4724.4  177.67  4809.5  178.28
  4930.8  178.75  4989.4  168.13    5030  169.06  5056.9  175.24  5089.4  177.37
  5132.8  175.99  5442.9  188.55  5624.1  206.37    5755  214.71  5894.6  217.13
    6313  231.03  6520.3  225.39  6641.2  229.15  6841.5  224.27  7180.7  237.52
#Mann= 12 ,-1 , 0
    1558     .16       0    2126     .05       0  2499.2     .12       0
  4724.4     .07       0  4809.5     .12       0  4930.8     .07       0
  4930.8     .07       0  5089.4     .07       0  5089.4     .12       0
  5132.8     .05       0  5894.6     .16       0    6313     .05       0
Bank Sta=4930.8,5089.4
XS Rating Curve= 0 ,0
Exp/Cntr=0.3,0.1

Type RM Length L Ch R = 1 ,115822  ,887,887,887
BEGIN DESCRIPTION:
NAVASOTA RIVER 250
END DESCRIPTION:
XS GIS Cut Line= 4
      3621984.38     10159285.24      3620663.68     10158369.53
      3617614.75     10156568.47      3616000.36     10156186.57
#Sta/Elev= 30
  3392.9  225.52  3727.1   214.5  3893.9  197.34  4056.2  189.65    4223  182.95
  4248.3  182.41  4934.9  178.17  4964.6  176.44  4985.6   167.7  5006.4  166.72
  5049.5  175.48  5102.3   177.6  5329.8  178.19    5440  178.19  5884.5  174.87
  5942.6  177.91  6561.6  179.48  6569.4  179.51  7497.9  184.97  8159.4  184.33
  8398.7  185.25  8745.4  188.46  8939.2  188.75  8982.1  185.51  9087.4  196.86
  9330.5  213.09  9678.5  216.19    9779  217.52  9790.4  217.62 10200.1  222.24
#Mann= 18 ,-1 , 0
  3392.9     .16       0  4056.2     .12       0    4223     .05       0
  4248.3     .12       0  4934.9     .07       0  5102.3     .12       0
  5329.8     .07       0    5440     .12       0  6561.6     .07       0
  6569.4     .12       0  8159.4     .07       0  8398.7     .12       0
  8745.4     .07       0  8939.2     .12       0  9087.4     .16       0
  9678.5     .05       0    9779     .16       0  9790.4     .05       0
#XS Ineff= 2 , 0
                         8964.86           189.2
Permanent Ineff=
       F       F
Bank Sta=4934.9,5102.3
XS Rating Curve= 0 ,0
Exp/Cntr=0.3,0.1

Type RM Length L Ch R = 1 ,114935  ,1909,1909,1909
BEGIN DESCRIPTION:
NAVASOTA RIVER 421
END DESCRIPTION:
XS GIS Cut Line= 3
      3622086.41     10159196.83      3618656.42     10155700.42
      3618049.09     10153635.51
#Sta/Elev= 30
  2661.5   224.2  3014.7  213.47    3625  184.81  3727.3  181.79  3836.7  179.23
  4909.9  175.36  4931.1  167.77  4945.2  171.16  5008.5   166.7  5044.2  167.96
  5065.4  175.14  5181.8     177  5327.1   172.7  6047.2  179.43    6128  179.81
  6161.7  179.97  6824.4  185.64  6829.9  186.17  7059.5  199.14  7172.8  199.37
  8214.8  204.09  8413.5  195.88  8579.6   206.8  8954.9  203.39  9005.9  215.48
    9139  215.57  9265.9  215.88  9346.3  215.76    9450  218.37  9711.8   221.9
#Mann= 18 ,-1 , 0
  2661.5     .16       0    3625     .05       0  3727.3     .16       0
  3836.7     .12       0  4909.9     .07       0  5065.4     .07       0
  5181.8     .12       0  6047.2     .07       0    6128     .12       0
  6161.7     .05       0  6824.4     .12       0  6829.9     .05       0
  7172.8     .16       0  8413.5     .05       0    9139      .1       0
  9265.9     .05       0  9346.3      .1       0    9450     .05       0
#XS Ineff= 2 , 0
       0                  8214.8       0  204.09
Permanent Ineff=
       F       F
Bank Sta=4909.9,5065.4
XS Rating Curve= 0 ,0
Exp/Cntr=0.3,0.1

Type RM Length L Ch R = 1 ,113026  ,1407,1407,1407
BEGIN DESCRIPTION:
NAVASOTA RIVER 420
END DESCRIPTION:
XS GIS Cut Line= 3
      3623776.66     10158875.01      3620784.91     10155919.11
      3618937.55     10153972.03
#Sta/Elev= 30
   794.3   211.6  1294.9  207.14  1478.7  209.31  1591.9  206.56  2051.5  207.79
  2221.2  203.64  2341.7  197.54  2645.5  183.22  2741.1  181.22    3197     177
  4420.4  178.18  4625.4  174.65  4922.4  176.08  4950.7  175.76    4979  166.75
  4998.2  166.11  5021.5  167.01  5042.6  176.96  5116.9  175.16    5230  175.47
  5790.3  178.88  5851.4  179.03  6040.1  179.07  6379.5  184.33  6591.8  198.87
  6620.1  203.85  6634.7  203.01  6655.3  199.48    6946   199.6    7684  219.73
#Mann= 11 ,-1 , 0
   794.3     .16       0  2341.7     .05       0  2741.1     .12       0
  4922.4     .07       0  5042.6     .12       0  5116.9     .07       0
    5230     .12       0  5790.3     .07       0  5851.4     .05       0
  6634.7     .16       0    6946     .05       0
Bank Sta=4922.4,5042.6
XS Rating Curve= 0 ,0
Exp/Cntr=0.3,0.1

Type RM Length L Ch R = 1 ,111619  ,2613,2613,2613
BEGIN DESCRIPTION:
NAVASOTA RIVER 419
END DESCRIPTION:
XS GIS Cut Line= 3
       3624608.7     10158825.61      3621779.66     10155233.73
      3619016.31     10153832.54
#Sta/Elev= 30
   427.8  212.38   968.8  205.65  1047.4  201.62  1475.6   207.1    1753  202.71
    2024  206.77  2320.7  198.45  2415.5  196.18    2572  193.37  2854.7  182.04
  3141.7  178.45  4658.7  175.91  4735.5  171.72  4942.4  175.07  4991.9   165.5
  5059.4  176.47  5135.8  176.21  5198.9  175.06  5477.8  178.07  5680.3  178.54
    6028  178.31  6050.3  175.61  6063.8  169.42  6094.8  168.65  6122.7  178.35
  6874.2  183.91  7119.1  194.59  7202.6  201.69  7351.8  200.44  8098.3  223.04
#Mann= 12 ,-1 , 0
   427.8     .16       0  2320.7      .1       0  2415.5     .16       0
    2572     .05       0  2854.7     .12       0  4942.4     .07       0
  5059.4     .12       0  5135.8     .07       0  5198.9     .12       0
  5477.8     .07       0  5680.3     .12       0  6063.8     .05       0
Bank Sta=4942.4,5059.4
XS Rating Curve= 0 ,0
Exp/Cntr=0.3,0.1

Type RM Length L Ch R = 1 ,109006  ,3855,3855,3855
BEGIN DESCRIPTION:
NAVASOTA RIVER 416
END DESCRIPTION:
XS GIS Cut Line= 4
      3626204.04     10158210.61      3621085.21     10153794.82
      3620689.91     10153305.16      3618785.59     10151969.55
#Sta/Elev= 30
 -2389.6  208.13 -2353.5  199.64 -2310.2  198.62 -1322.5  198.65 -1128.5  198.76
  -750.3  196.59  -664.4  195.56  -426.5  196.08   -17.9  199.78   534.9  190.49
   807.8  180.56  3310.4  177.68  4681.4  176.22  4937.3   175.2  4978.7  164.12
  5015.2  166.03  5036.2  180.75  5754.6  201.65  5970.5  213.62  6358.6  211.78
  6393.3  210.23  6429.3  198.18  6443.8  198.26  6458.6  205.66  6550.1  211.72
  6695.1  216.82  7134.1  217.88    7176  224.86  7250.5  222.74    7326  224.95
#Mann= 18 ,-1 , 0
 -2389.6     .05       0 -2310.2     .16       0 -1322.5      .1       0
 -1128.5     .16       0  -750.3     .05       0  -664.4     .16       0
  -426.5     .16       0   -17.9     .16       0   534.9     .05       0
   807.8     .12       0  3310.4     .07       0  4681.4     .03       0
  5036.2     .05       0  6358.6     .16       0  6429.3     .12       0
  6550.1     .16       0  6695.1     .05       0  7250.5      .1       0
Bank Sta=4681.4,5036.2
XS Rating Curve= 0 ,0
Exp/Cntr=0.3,0.1

Type RM Length L Ch R = 1 ,105151  ,2999,2999,2999
BEGIN DESCRIPTION:
NAVASOTA RIVER 415
END DESCRIPTION:
XS GIS Cut Line= 4
      3627886.86     10155345.82      3625407.71     10154158.33
      3621907.71     10153533.33      3618900.98     10151800.83
#Sta/Elev= 30
  -497.7  216.73  -159.8  217.13   192.9  198.52   361.9  176.91  1178.4   184.5
    1421  198.45  1641.7  197.99  1698.5  190.94  1749.1  195.36  1932.1  200.12
  2683.5  200.27  2976.1  191.68  3126.3  186.34  3306.3  182.66  3831.6  180.89
  3898.3  180.67  4867.5  177.41  4987.6  159.98    5091  176.07  5815.1  175.53
  5928.4     167  6023.4   175.8  7283.3  187.89  8162.5  214.14  8461.2  214.85
  8527.1  213.04  8607.9  204.22  8704.2  213.57  9216.4  223.61  9276.7  223.68
#Mann= 17 ,-1 , 0
  -497.7     .16       0   192.9     .12       0  1178.4     .05       0
  1641.7     .08       0  1749.1     .05       0  1932.1     .16       0
  2976.1     .05       0  3126.3     .16       0  3306.3     .12       0
  3831.6     .05       0  3898.3     .12       0  4867.5     .07       0
    5091     .12       0  5815.1     .05       0  8461.2     .16       0
  8527.1     .05       0  9216.4     .08       0
#XS Ineff= 2 , 0
         2683.56  200.09
Permanent Ineff=
       F       F
Bank Sta=4867.5,5091
XS Rating Curve= 0 ,0
Exp/Cntr=0.3,0.1

Type RM Length L Ch R = 1 ,102152  ,1823,1823,1823
BEGIN DESCRIPTION:
NAVASOTA RIVER 252
END DESCRIPTION:
XS GIS Cut Line= 3
      3629505.13     10155249.88      3622044.86     10151463.02
      3619722.78     10150117.51
#Sta/Elev= 30
 -2759.4  215.66 -2680.7  210.64 -2573.2  197.55 -1858.8  184.87 -1827.6  192.36
 -1805.9  185.03  -333.7  181.75  -311.2  171.89  -221.5  182.08   654.9  180.97
  1394.4  192.64  1502.9  189.96  2588.1  186.51  2696.6  182.78  3300.1  178.33
  3794.5  177.25  4889.3  174.03    5006  159.39  5089.7  174.59  5923.4  180.48
  5991.5  191.61  6296.3  188.04    6402  191.46    6713   191.4  6822.5  191.41
  6953.7  196.19  7523.1  212.69  7746.2  213.52  7877.4   209.1  8290.7  218.96
#Mann= 19 ,-1 , 0
 -2759.4     .08       0 -2680.7     .05       0 -1805.9     .12       0
   654.9     .05       0  1394.4     .08       0  1502.9     .05       0
  2588.1     .16       0  2696.6     .12       0  3300.1     .05       0
  3794.5     .12       0  4889.3     .07       0  5089.7     .05       0
  6296.3     .07       0    6402     .16       0    6713     .12       0
  6822.5     .16       0  6953.7     .05       0  7523.1     .08       0
  7746.2     .05       0
#XS Ineff= 2 , 0
         1415.82  194.56
Permanent Ineff=
       F       F
Bank Sta=4889.3,5089.7
XS Rating Curve= 0 ,0
Exp/Cntr=0.3,0.1

Type RM Length L Ch R = 1 ,100329  ,6477,6477,6477
BEGIN DESCRIPTION:
NAVASOTA RIVER 251
END DESCRIPTION:
XS GIS Cut Line= 3
      3632380.12     10152786.57      3626016.21     10151788.54
      3621339.45     10149399.98
#Sta/Elev= 30
   -4407  230.16 -3566.1  195.29 -1856.3  189.37  -451.2  197.95    43.2   176.7
   234.4  175.28   303.6  186.29   401.5  169.13     539  176.51     756  178.72
    2414  184.54  2480.7  195.07  2519.5  185.04  3312.2  179.94  3517.5  177.02
  3558.5  176.09  3615.6  175.22  3688.6   174.2  4947.5  173.19    4980  158.97
  5113.6  173.57  5245.2  169.94  5353.8  175.74  5384.8  176.04  6463.5  186.13
  6813.4  199.59  6946.8  213.84  7013.6  203.73    7176  235.58  7286.1  239.97
#Mann= 19 ,-1 , 0
   -4407     .05       0 -1856.3     .16       0  -451.2     .12       0
    43.2     .05       0   234.4     .12       0   401.5     .07       0
     539     .12       0     756     .05       0  3312.2     .12       0
  3517.5     .05       0  3558.5     .12       0  3615.6     .05       0
  3688.6     .12       0  4947.5     .07       0  5113.6     .12       0
  5245.2     .07       0  5353.8     .12       0  5384.8     .05       0
    7176      .1       0
#XS Ineff= 2 ,-1
 -3957.1  -598.7  201.55  -598.7    2466  195.06
Permanent Ineff=
       F       F
Bank Sta=4947.5,5113.6
XS Rating Curve= 0 ,0
Exp/Cntr=0.3,0.1
