--- HOLMAN CREEK.prj (project) ---

Proj Title=HOLMAN CREEK Base Level Engineering
Current Plan=p01
Default Exp/Contr=0.3,0.1
English Units
Geom File=g01
Flow File=f01
Plan File=p01
Y Axis Title=Elevation
X Axis Title(PF)=Main Channel Distance
X Axis Title(XS)=Station
BEGIN DESCRIPTION:
HOLMAN CREEK
END DESCRIPTION:
DSS Export Rating Curves= 0
DSS Export Rating Curve Sorted= 0
DSS Export Volume Flow Curves= 0
DXF OffsetX= 0
DXF OffsetY= 0
DXF ScaleX= 1
DXF ScaleY= 10

--- HOLMAN CREEK.p01 (plan) ---

Plan Title=Multiple Run
Short Identifier=Multiple
Geom File=g01
Flow File=f01
Subcritical Flow
K Sum by GR= 0
Std Step Tol= 0.01
Critical Tol= 0.01
Num of Std Step Trials= 20
Max Error Tol= 0.3
Flow Tol Ratio= 0.001
Split Flow NTrial= 30
Split Flow Tol= 0.02
Split Flow Ratio= 0.02
Log Output Level= 0
Friction Slope Method= 1
Unsteady Friction Slope Method= 2
Unsteady Bridges Friction Slope Method= 1
Parabolic Critical Depth
Global Vel Dist=  1 , 1 , 1
Global Log Level= 0
CheckData=True
Encroach Param= -1, 0, 0, 0
BEGIN DESCRIPTION:
Multiple Run
END DESCRIPTION:

--- HOLMAN CREEK.f01 (steady flow) ---

Flow Title=Multiple
Program Version=4.10
Number of Profiles= 7
Profile Names=10-year,25-year,50-year,1pct_min,100-year,1pct_plu,500-year
River Rch & RM=HOLMAN CREEK,Reach-1         ,52737
     893    1212    1471    1303    1762    2383    2520
River Rch & RM=HOLMAN CREEK,Reach-1         ,50636
    1417    1961    2412    2160    2921    3950    4272
River Rch & RM=HOLMAN CREEK,Reach-1         ,44476
    1500    2081    2564    2299    3110    4205    4563
River Rch & RM=HOLMAN CREEK,Reach-1         ,42156
    2560    3629    4534    4116    5566    7527    8370
River Rch & RM=HOLMAN CREEK,Reach-1         ,37944
    2637    3738    4671    4239    5732    7752    8618
River Rch & RM=HOLMAN CREEK,Reach-1         ,36789
    2884    4101    5133    4666    6311    8534    9518
River Rch & RM=HOLMAN CREEK,Reach-1         ,34050
    2899    4120    5156    4685    6336    8569    9551
River Rch & RM=HOLMAN CREEK,Reach-1         ,33665
    3081    4398    5521    5032    6805    9204   10320
River Rch & RM=HOLMAN CREEK,Reach-1         ,30842
    3443    4926    6192    5648    7639   10330   11603
River Rch & RM=HOLMAN CREEK,Reach-1         ,16523
    7375   10731   13644   12559   16985   22970   26263
River Rch & RM=HOLMAN CREEK,Reach-1         ,12525
    8664   12662   16149   14908   20161   27265   31345
River Rch & RM=HOLMAN CREEK,Reach-1         ,9592
    8630   12597   16053   14806   20024   27080   31079
River Rch & RM=HOLMAN CREEK,Reach-1         ,7573
   10849   15920   20363   18845   25485   34466   39809
Boundary for River Rch & Prof#=HOLMAN CREEK,Reach-1         , 1
Up Type= 0
Dn Type= 1
Dn Known WS=397.08
Boundary for River Rch & Prof#=HOLMAN CREEK,Reach-1         , 2
Up Type= 0
Dn Type= 1
Dn Known WS=398.53
Boundary for River Rch & Prof#=HOLMAN CREEK,Reach-1         , 3
Up Type= 0
Dn Type= 1
Dn Known WS=399.75
Boundary for River Rch & Prof#=HOLMAN CREEK,Reach-1         , 4
Up Type= 0
Dn Type= 1
Dn Known WS=399.34
Boundary for River Rch & Prof#=HOLMAN CREEK,Reach-1         , 5
Up Type= 0
Dn Type= 1
Dn Known WS=401.08
Boundary for River Rch & Prof#=HOLMAN CREEK,Reach-1         , 6
Up Type= 0
Dn Type= 1
Dn Known WS=403.1
Boundary for River Rch & Prof#=HOLMAN CREEK,Reach-1         , 7
Up Type= 0
Dn Type= 1
Dn Known WS=404.22
DSS Import GetInterval= 0
DSS Import GetPeak= 0
DSS Import FillOption= 0

--- HOLMAN CREEK.g01 (geometry) ---

Geom Title=Existing Conditions
Program Version=4.10

River Reach=HOLMAN CREEK    ,Reach-1
Reach XY= 30
      3542101.13     10595211.36      3541697.19     10593851.95
      3542030.98     10593457.09        3540739.     10590741.24
      3541532.97      10589766.5      3542222.78     10586573.62
      3542105.88     10584945.14      3543052.11     10581931.64
      3542798.99     10580438.12      3542182.28     10580096.75
      3542662.32     10578907.51       3542205.6       10576223.
      3542793.88     10576058.17      3543941.49     10573871.08
      3544071.11     10571632.05      3543703.24     10571193.36
      3544486.32     10570001.64      3544093.81     10569596.11
      3544099.43     10567907.42      3543431.18     10567675.25
      3543801.74     10567336.57      3543493.84     10566797.47
      3544093.37     10566376.21      3544631.86     10566621.99
      3546340.94     10564236.12      3546472.12     10561711.87
      3546047.49     10560349.42      3546599.53     10558827.31
      3545544.05     10557325.47      3546002.11     10556211.64

Type RM Length L Ch R = 1 ,52737   ,642,642,642
BEGIN DESCRIPTION:
HOLMAN CREEK 74.0
END DESCRIPTION:
XS GIS Cut Line= 2
      3542996.44     10594936.27      3541345.43     10595210.28
#Sta/Elev= 30
    4094   497.9  4216.7  491.81    4258  490.32  4321.4  488.82  4343.7  489.05
  4365.6  487.84  4460.5  484.78  4574.8  483.75  4615.4  484.04  4678.7  482.93
  4797.8  481.18  4831.3  481.96  4899.2  480.69  4909.3  479.98  4942.6  479.93
  4980.3   479.8  4990.4   477.8  4997.6  475.36  5000.3  474.86  5003.6  475.36
    5009  478.21  5020.8   479.7    5031  479.03  5072.1  480.65  5172.9  481.31
  5274.3  483.77  5374.9  484.93  5557.6  487.35    5607  488.88  5767.6  491.17
#Mann= 10 ,-1 , 0
    4094     .05       0    4258     .08       0  4365.6     .05       0
  4678.7     .16       0  4942.6     .12       0  4997.6     .07       0
  5003.6     .12       0  5072.1     .16       0  5374.9      .1       0
    5607     .05       0
Bank Sta=4980.3,5020.8
XS Rating Curve= 0 ,0
Exp/Cntr=0.3,0.1

Type RM Length L Ch R = 1 ,52095   ,588,588,588
BEGIN DESCRIPTION:
HOLMAN CREEK 72.0
END DESCRIPTION:
XS GIS Cut Line= 2
      3543568.71      10594137.5      3540082.55     10595012.51
#Sta/Elev= 30
  3461.1  492.83  3818.5  491.36  3948.9  490.07  4055.6  490.92  4198.4  488.87
  4301.4  486.66  4365.7  485.28  4401.7  483.44  4602.5  481.02  4879.1  479.11
  4911.7   479.1  4952.6  479.35  4983.5  477.73  5001.1  475.51  5003.9  475.01
  5007.1  475.51  5019.1  476.07  5024.7  477.29  5125.4  478.35  5384.3  480.51
  5801.1  486.51  5842.2  486.05  5878.2  486.63  6140.1  486.76  6282.6  486.73
  6377.3  487.92  6591.9  486.96  6849.7  489.89  7010.9  490.76  7055.4   491.3
#Mann= 11 ,-1 , 0
  3461.1     .05       0  4198.4     .08       0  4301.4     .05       0
  4602.5     .16       0  4879.1     .12       0  4911.7     .16       0
  5001.1     .07       0  5007.1     .16       0  5125.4     .05       0
  6140.1      .1       0  7010.9     .16       0
Bank Sta=4983.5,5024.7
XS Rating Curve= 0 ,0
Exp/Cntr=0.3,0.1

Type RM Length L Ch R = 1 ,51507   ,871,871,871
BEGIN DESCRIPTION:
HOLMAN CREEK 71.0
END DESCRIPTION:
XS GIS Cut Line= 2
      3542992.28     10593873.62      3539797.83     10594408.34
#Sta/Elev= 30
  3762.7  489.37  3854.1  489.39  3987.3  486.27  4004.2  485.26  4290.1  479.35
    4719  479.04  4774.4  478.46    4896  477.18  4969.4  476.82  5006.1  475.21
  5017.1  475.19  5019.9  474.69  5023.1  475.19  5054.3  476.63  5097.9  477.67
  5189.2   479.7  5357.1  481.12  5486.5  481.55  5600.6  480.39  5638.6  478.51
  5735.7  479.03  5750.1  478.12  5777.7  479.88    5811  479.75  5838.4   481.9
  5942.9  482.35  5967.1  482.48  6180.3  484.16  6226.7  485.84  7001.6  491.82
#Mann= 16 ,-1 , 0
  3762.7     .05       0  3987.3     .08       0  4004.2     .05       0
    4719     .16       0  4774.4     .05       0    4896      .1       0
  5006.1     .16       0  5017.1     .07       0  5023.1     .16       0
  5097.9     .05       0  5189.2     .16       0  5357.1     .05       0
  5735.7     .12       0  5942.9     .05       0  5967.1     .12       0
  6180.3     .05       0
Bank Sta=4969.4,5054.3
XS Rating Curve= 0 ,0
Exp/Cntr=0.3,0.1

Type RM Length L Ch R = 1 ,50636   ,685,685,685
BEGIN DESCRIPTION:
HOLMAN CREEK 70.0
END DESCRIPTION:
XS GIS Cut Line= 4
      3544050.27     10593539.74      3542231.71     10593431.23
       3541120.6     10593639.57      3539455.53     10593908.41
#Sta/Elev= 30
  2974.7  500.12  3028.3  499.48  3140.4  497.31  3328.4  494.45  3825.4  486.43
  3957.3  484.62  4069.8  484.42  4104.9  483.04  4144.9  477.43  4214.4   480.8
  4337.7  482.55  4436.6  481.14  4535.4  480.45  4728.2   479.2  4933.9  478.57
  4969.1  477.84  4979.2   475.5  4986.5  470.91  4996.6  469.48  4999.3  468.98
  5002.6  469.48  5019.9  472.43  5073.3  470.98  5096.7  474.22  5339.8  476.35
  5531.4  477.49  6257.9  482.72  6440.8  484.49  7019.3  489.99  7613.6  495.92
#Mann= 20 ,-1 , 0
  2974.7     .16       0  3028.3     .12       0  3140.4     .16       0
  3328.4     .05       0  3825.4     .16       0  3957.3     .05       0
  4069.8     .16       0  4214.4     .05       0  4337.7     .12       0
  4436.6      .1       0  4535.4     .05       0  4728.2     .05       0
  4996.6     .07       0  5002.6     .16       0  5073.3     .12       0
  5339.8     .05       0  5531.4     .05       0  6257.9      .1       0
  6440.8     .05       0  7019.3     .05       0
Bank Sta=4979.2,5019.9
XS Rating Curve= 0 ,0
Exp/Cntr=0.3,0.1

Type RM Length L Ch R = 1 ,49951   ,1015,1015,1015
BEGIN DESCRIPTION:
HOLMAN CREEK 69.0
END DESCRIPTION:
XS GIS Cut Line= 2
      3543746.43     10592415.62      3539831.51      10593630.9
#Sta/Elev= 30
  2768.9  505.99  3286.5  495.56  3736.7  492.11  3984.7  484.33  4145.1   480.9
  4458.1  478.84  4797.2  473.82  4900.8  474.42  4951.3  472.24  4960.7  470.03
  4965.9  467.18  4972.3  469.26  4982.7   468.8  4993.2  467.05  4995.5   465.4
  4998.3   464.9  5001.5   465.4  5014.2   469.2  5036.3  472.35  5075.8  473.85
  5103.7  474.08  5286.4  476.17  5334.7   472.4    5412  476.35  5470.2  477.33
  5987.9  482.04  6077.4  484.68  6562.8  488.19  6669.5  489.37  6868.1  491.28
#Mann= 9 ,-1 , 0
  2768.9     .05       0  4458.1     .16       0  4797.2     .12       0
  4995.5     .07       0  5001.5     .12       0  5075.8     .16       0
  5103.7     .05       0  6562.8      .1       0  6669.5     .05       0
Bank Sta=4951.3,5036.3
XS Rating Curve= 0 ,0
Exp/Cntr=0.3,0.1

Type RM Length L Ch R = 1 ,48936   ,1366,1366,1366
BEGIN DESCRIPTION:
HOLMAN CREEK 67.0
END DESCRIPTION:
XS GIS Cut Line= 2
      3542744.37     10591652.09      3539890.23     10593034.03
#Sta/Elev= 30
  3290.2  491.05  3598.6   483.4  3779.3  485.53  3959.4  485.18    4084  483.17
  4437.1  473.62    4609  471.21  4670.4  471.63  4692.6  473.04  4699.3  471.01
  4727.8  470.75  4759.3  472.39  4789.6  469.79  4908.1  468.72  4937.1  469.62
  4970.3  467.92  4981.5  468.81  4992.6   467.3  4998.4  462.76    5001  462.45
  5003.8  461.95    5007  462.45    5021  469.41    5064  470.64    5176  474.02
  5607.8  478.07  5624.2  478.99    5788  482.37  6240.2  488.56  6461.3  493.95
#Mann= 9 ,-1 , 0
  3290.2     .05       0  4727.8     .12       0    5001     .07       0
    5007     .12       0    5064     .16       0    5176     .05       0
  5607.8     .16       0  5624.2     .12       0    5788     .05       0
Bank Sta=4981.5,5021
XS Rating Curve= 0 ,0
Exp/Cntr=0.3,0.1

Type RM Length L Ch R = 1 ,47570   ,896,896,896
BEGIN DESCRIPTION:
HOLMAN CREEK 65.0
END DESCRIPTION:
XS GIS Cut Line= 3
      3542622.62     10590970.45      3540638.29     10591621.48
      3540076.59     10592006.34
#Sta/Elev= 30
  3235.6  490.25    3394  486.01  3709.8  479.85  3996.2   477.8  4219.4  474.88
  4307.6  475.35  4556.7  471.94  4641.3  470.45  4650.4  470.09    4678  468.61
  4746.8  467.83  4867.4  465.83  4883.5  464.67  4941.1  466.45  4982.8  464.78
  4990.7  460.36  4993.5  459.86  4996.7  460.36  5004.2  461.13  5019.9  465.36
  5046.3  465.22  5077.9  467.31  5168.6  467.18  5267.4   467.8  5371.2  470.09
  5527.9  475.88  5646.1  481.42  5742.1  483.44  5852.7  485.68  6004.9  485.21
#Mann= 13 ,-1 , 0
  3235.6     .05       0  4219.4      .1       0  4307.6     .05       0
  4556.7      .1       0  4641.3     .05       0  4650.4      .1       0
  4746.8     .05       0  4883.5     .16       0  4990.7     .07       0
  4996.7     .16       0  5168.6     .05       0  5527.9     .16       0
  5742.1     .05       0
Bank Sta=4982.8,5019.9
XS Rating Curve= 0 ,0
Exp/Cntr=0.3,0.1

Type RM Length L Ch R = 1 ,46674   ,930,930,930
BEGIN DESCRIPTION:
HOLMAN CREEK 62.0
END DESCRIPTION:
XS GIS Cut Line= 4
      3542774.24     10590705.54      3540959.49     10590928.77
       3540495.6     10590874.81      3539449.55     10590874.81
#Sta/Elev= 30
  3027.5  496.81  3452.8  486.79  3734.9   487.1  3805.5  485.22    4007  474.78
  4037.2  476.83    4097  475.67  4127.9  476.73    4148  475.28  4269.6  477.73
  4753.4  467.75  4958.8  464.42  4984.2  463.08  5001.3  458.61  5004.1  458.11
  5007.3  458.61  5024.4  462.88  5048.5  463.94  5064.7  461.98  5155.3  466.54
  5301.7  467.45  5404.2  469.04  5439.5  469.97  5516.4  472.18  5596.4  471.47
  5778.8  474.44  5812.8  474.79  6006.4  476.53  6176.4  480.61    6369  482.94
#Mann= 10 ,-1 , 0
  3027.5     .05       0  4753.4     .16       0  4958.8     .12       0
  5001.3     .07       0  5007.3     .12       0  5301.7     .05       0
  5404.2     .12       0  5439.5     .05       0  5778.8     .16       0
  5812.8     .05       0
#XS Ineff= 2 , 0
         4238.92  477.91
Permanent Ineff=
       F       F
Bank Sta=4984.2,5024.4
XS Rating Curve= 0 ,0
Exp/Cntr=0.3,0.1

Type RM Length L Ch R = 1 ,45744   ,1103,1103,1103
BEGIN DESCRIPTION:
HOLMAN CREEK 61.0
END DESCRIPTION:
XS GIS Cut Line= 3
      3542336.21     10589939.18       3540273.7     10590543.35
      3539461.23     10590621.48
#Sta/Elev= 30
    3527  491.13  3594.1   489.5  3820.7  478.97  3983.7  473.06  4015.9  470.42
    4160  468.07  4198.6  468.66    4232  466.53  4260.2  467.42  4298.9   465.3
  4370.9  464.15  4442.9  465.08  4841.1  461.65  4936.8  463.03  4974.4  462.05
  4975.5  462.05  4997.5   456.6  5000.3   456.1  5003.5   456.6  5021.4  462.94
  5052.7  463.11  5104.7  460.99  5323.6  465.44    5459  465.97  5538.5  468.63
  5674.4  472.07  5848.6  471.69  6109.8  474.97  6341.6  479.69  6492.4  480.54
#Mann= 8 ,-1 , 0
    3527     .05       0  3820.7      .1       0  3983.7     .05       0
  4841.1     .16       0  4974.4     .12       0  4997.5     .07       0
  5003.5     .12       0  5538.5     .05       0
Bank Sta=4975.5,5021.4
XS Rating Curve= 0 ,0
Exp/Cntr=0.3,0.1

Type RM Length L Ch R = 1 ,44641   ,36,36,36
BEGIN DESCRIPTION:
HOLMAN CREEK 60.0
END DESCRIPTION:
XS GIS Cut Line= 3
      3542825.57     10589304.65      3541266.58     10589787.28
      3539679.77     10590328.95
#Sta/Elev= 30
    3655  491.06  3863.3   486.8  3966.8  485.35    4135  479.95  4244.8  478.35
  4343.4  479.02  4433.3  479.65  4569.4     476  4869.4  463.91  4976.4  460.71
  4981.7  459.99  4988.1  456.63  4995.6  455.65  4998.3  455.15  5001.6  455.65
  5014.3  458.37    5030  458.62  5040.4  460.74  5112.1  459.42    5334  460.79
  5405.7  463.59  5619.3     467  5774.5  466.66  6060.2  469.28  6137.2  469.65
  6304.5  469.95  6518.7  470.91  6679.6  472.05  6865.4  475.96  6963.7  478.13
#Mann= 12 ,-1 , 0
    3655     .08       0  3863.3     .05       0  4343.4     .08       0
  4869.4     .05       0  4995.6     .04       0  5001.6     .05       0
  5774.5     .08       0  6060.2     .05       0  6137.2     .08       0
  6304.5     .05       0  6518.7     .08       0  6865.4     .05       0
Bank Sta=4976.4,5040.4
XS Rating Curve= 0 ,0
Exp/Cntr=0.3,0.1

Type RM Length L Ch R = 1 ,44605   ,129,129,129
BEGIN DESCRIPTION:
HOLMAN CREEK 59.0
END DESCRIPTION:
XS GIS Cut Line= 2
      3542815.24      10589245.6      3539656.29     10590283.54
#Sta/Elev= 30
  3651.6  488.84  3657.6  489.73  3684.1  488.15  3721.2  488.59  3747.7  486.63
  3882.8  485.47  4039.2  480.99  4108.1  480.59  4134.7  478.02  4147.5  479.28
  4267.2  477.89  4420.9  479.82  4484.5  479.22  4489.8  478.05  4548.1  477.15
  4889.7  463.76  4972.2   460.9  4995.7  455.47  4998.5  454.97  5001.7  455.47
  5030.5  461.14  5139.1  458.95  5353.8  460.89  5422.6  462.75  5640.1  467.34
  5791.7  466.71  6083.7  469.37  6112.1  469.53  6654.8  471.95  6976.7  478.44
#Mann= 9 ,-1 , 0
  3651.6     .08       0  3882.8     .05       0  4147.5     .08       0
  4889.7     .05       0  4995.7     .04       0  5001.7     .05       0
  5422.6     .08       0  6083.7     .05       0  6112.1     .08       0
Bank Sta=4972.2,5030.5
XS Rating Curve= 0 ,0
Exp/Cntr=0.3,0.1

Type RM Length L Ch R = 1 ,44476   ,80,80,80
BEGIN DESCRIPTION:
HOLMAN CREEK 58.0
END DESCRIPTION:
XS GIS Cut Line= 2
      3542835.98     10589117.15      3539617.31     10590151.85
#Sta/Elev= 30
    3613  486.92  3643.7  485.17  3745.2  484.41  3816.6  481.18  4066.1  475.04
  4071.4  476.16  4098.2  474.96  4257.8  474.42  4301.3  476.66  4397.6  478.48
  4493.9  477.33  4691.7  472.15  4961.6   459.8  4993.1  455.04  5012.6  456.79
  5014.9   454.8  5017.6   454.3  5020.9   454.8  5035.1  458.97  5098.1  460.65
  5161.2  460.43  5255.7  456.44  5297.7  459.52  5518.3  464.83  5536.6     464
  5791.4  468.29  6290.5  469.88  6579.2  472.72  6916.1  478.48  6993.9  478.32
#Mann= 3 ,-1 , 0
    3613     .08       0  5014.9     .07       0  5020.9     .08       0
Bank Sta=4961.6,5035.1
XS Rating Curve= 0 ,0
Exp/Cntr=0.3,0.1

Type RM Length L Ch R = 1 ,44396   ,986,986,986
BEGIN DESCRIPTION:
HOLMAN CREEK 57.0
END DESCRIPTION:
XS GIS Cut Line= 4
      3542822.14     10589068.53      3541669.36     10589460.89
        3541402.     10589481.72      3539679.79     10590085.88
#Sta/Elev= 30
  3663.6  485.39  3814.9  482.19  4029.1  475.06  4123.2  473.26  4297.4  473.94
  4424.2  478.23    4551  476.58  4745.2  471.54  4968.8  461.05  4995.9  455.64
  4998.7  455.14  5001.9  455.64    5009     456    5019  458.93    5029  460.15
  5099.2  458.84  5191.3   459.6  5257.8  460.36  5276.5  458.63  5283.5  456.14
  5297.6  455.72  5314.5     458  5342.5  458.18  5526.2  463.66  5588.2  463.81
    5817  468.54  5986.6  467.82    6187  468.67  6796.5  474.52  6974.6  477.41
#Mann= 6 ,-1 , 0
  3663.6     .08       0  4995.9     .07       0  5001.9     .08       0
  5191.3     .16       0  5297.6     .12       0  5342.5     .08       0
Bank Sta=4968.8,5029
XS Rating Curve= 0 ,0
Exp/Cntr=0.3,0.1

Type RM Length L Ch R = 1 ,43410   ,1254,1254,1254
BEGIN DESCRIPTION:
HOLMAN CREEK 56.0
END DESCRIPTION:
XS GIS Cut Line= 2
      3542765.64     10588485.96      3540390.68     10588991.16
#Sta/Elev= 30
  3628.5  481.38  3797.8  475.99  3810.2  475.73  3959.3  472.72  4115.1  467.04
    4204  465.67  4303.2  462.08  4429.6  459.93  4446.9  461.64  4466.9   459.3
  4531.8  458.84  4552.2  461.65  4572.7  458.43  4621.1  457.66  4882.9  456.72
  4982.1   456.6  4991.9  455.13  5009.3  454.91  5012.1  454.41  5015.3  454.91
    5043  456.77  5221.6  460.38  5358.4  464.28  5584.8  464.47  5707.5  468.45
  5901.8  468.24  5922.2  469.85  5938.2  473.23  5993.8  474.81  6056.6  474.33
#Mann= 9 ,-1 , 0
  3628.5     .05       0  3797.8      .1       0  3810.2     .05       0
  4466.9     .16       0  4621.1     .05       0  4882.9     .16       0
  5009.3     .07       0  5015.3     .16       0  5221.6     .05       0
#XS Ineff= 2 , 0
          4551.7   461.7
Permanent Ineff=
       F       F
Bank Sta=4982.1,5043
XS Rating Curve= 0 ,0
Exp/Cntr=0.3,0.1

Type RM Length L Ch R = 1 ,42156   ,1005,1005,1005
BEGIN DESCRIPTION:
HOLMAN CREEK 55.0
END DESCRIPTION:
XS GIS Cut Line= 4
      3542726.47     10587910.39      3541927.89     10587749.81
      3541506.89     10587814.92      3539258.62     10586799.29
#Sta/Elev= 30
  3996.7  483.62  4270.4  477.32  4372.1  473.81    4423   471.6  4468.8  467.13
  4531.6  462.92    4620  460.42  4626.4  460.02  4677.3  456.88  4723.1  456.03
    4779  455.68  4848.2  456.97  4877.8  457.14  4913.8  455.25  4955.8  454.54
  4958.5  454.04  4961.8  454.54  5014.5  454.57  5500.3  456.44  5604.6   459.4
  5700.5  463.51  5822.4   463.6  6111.2  462.96    6281  464.12  6343.9  464.05
  6494.2  465.06  7033.6  469.99  7298.9  473.62  7448.6  477.59  7704.3  482.32
#Mann= 12 ,-1 , 0
  3996.7     .05       0    4620     .16       0  4848.2     .12       0
  4913.8     .16       0  4955.8     .07       0  4961.8     .16       0
  5014.5     .12       0  5700.5     .05       0  5822.4     .12       0
    6281     .05       0  6343.9     .12       0  6494.2     .05       0
Bank Sta=4626.4,5604.6
XS Rating Curve= 0 ,0
Exp/Cntr=0.3,0.1

Type RM Length L Ch R = 1 ,41151   ,511,511,511
BEGIN DESCRIPTION:
HOLMAN CREEK 54.0
END DESCRIPTION:
XS GIS Cut Line= 2
       3542644.7     10587499.85      3540882.55     10586440.82
#Sta/Elev= 30
  4250.7  484.28  4405.4  481.29  4433.1  480.11  4506.9  475.88  4549.7  474.46
  4586.6  470.19    4608  469.51  4687.6  464.78  4703.2  462.89  4720.2  461.82
  4724.5  461.98  4755.4     459  4832.9  455.66    4878  454.55  5047.1  455.04
    5182  454.33  5184.7  453.83    5188  454.33  5227.7  454.57  5301.6  457.31
  5408.8   457.6  5460.9  456.21  5635.8  459.53  5746.5  461.42  5905.8  461.12
  6028.2  463.12  6123.4  466.08  6190.4  469.91  6261.4  472.91  6306.6  473.97
#Mann= 5 ,-1 , 0
  4250.7     .05       0  4720.2     .12       0  4832.9     .05       0
    5182    .033       0    5188     .05       0
Bank Sta=4755.4,5635.8
XS Rating Curve= 0 ,0
Exp/Cntr=0.3,0.1

Type RM Length L Ch R = 1 ,40640   ,930,930,930
BEGIN DESCRIPTION:
HOLMAN CREEK 52.0
END DESCRIPTION:
XS GIS Cut Line= 4
      3542648.41      10587185.6      3542205.67     10586816.65
      3541901.85     10586491.13      3540926.24     10586239.64
#Sta/Elev= 30
  4235.2  481.04  4263.9  481.05  4420.1  477.63  4483.9  473.37    4562  467.02
  4576.3  464.82  4618.8  461.95  4640.1  460.74  4646.9  459.65  4654.4  458.26
  4743.4  454.66  4786.8  454.54  4789.5  454.04  4792.8  454.54    5023  454.77
  5263.2  456.24  5395.2  456.61  5517.5  458.12  5576.7  459.69  5675.1  461.38
  5873.3  461.25  5969.1  463.34  5990.1  464.45  6030.9  465.62  6091.2  468.69
  6134.3   470.5  6175.6  473.66  6216.9  474.65  6239.5  476.07  6264.3  475.48
#Mann= 9 ,-1 , 0
  4235.2     .05       0  4618.8     .12       0  4743.4     .05       0
  4786.8    .033       0  4792.8     .05       0  5263.2     .16       0
  5395.2     .05       0  5990.1     .08       0  6091.2     .05       0
Bank Sta=4646.9,5576.7
XS Rating Curve= 0 ,0
Exp/Cntr=0.3,0.1

Type RM Length L Ch R = 1 ,39710   ,681,681,681
BEGIN DESCRIPTION:
HOLMAN CREEK 51.0
END DESCRIPTION:
XS GIS Cut Line= 3
      3542941.22     10585799.96      3542240.39     10585792.35
      3540942.08     10586191.65
#Sta/Elev= 30
  4137.6  479.92  4210.1   478.4  4436.7  473.01  4596.7  465.49  4626.7     463
  4656.7   459.3  4664.1  458.67  4733.7   454.6  4736.5   454.1  4739.7   454.6
  5157.5  456.78  5162.7  455.45  5190.2  456.15  5195.4  455.18  5276.1  455.09
  5293.5  456.11  5298.8  455.68  5326.2  457.74  5331.5  456.65  5349.3   458.3
  5396.9  459.28  5429.6  460.74  5558.6  460.42  5772.3  462.38  5810.2  463.58
  5851.5  463.22  6018.9  467.88  6032.2  468.86    6137  474.29  6196.8  475.71
#Mann= 7 ,-1 , 0
  4137.6     .08       0  4210.1     .16       0  4664.1     .05       0
  4733.7    .033       0  4739.7     .05       0  6032.2     .08       0
    6137     .05       0
#XS Ineff= 2 , 0
                         5461.65          460.96
Permanent Ineff=
       F       F
Bank Sta=4656.7,5396.9
XS Rating Curve= 0 ,0
Exp/Cntr=0.3,0.1

Type RM Length L Ch R = 1 ,39029   ,1085,1085,1085
BEGIN DESCRIPTION:
HOLMAN CREEK 49.0
END DESCRIPTION:
XS GIS Cut Line= 2
      3542935.52     10585351.16      3540176.11     10584769.77
#Sta/Elev= 30
  4116.4  476.53  4154.7  474.69    4171  474.09  4191.7  471.21    4263  469.33
  4281.1  467.87  4286.2  466.16  4365.2  458.72  4380.7   457.2  4427.1  454.72
  4443.9  454.59  4446.7  454.09  4449.9  454.59  4674.4  455.22  5374.9   454.7
  5438.2  454.62  5560.9  458.52  5582.8  458.81  5652.8  458.96  5789.1   456.7
  5928.3  458.16  5990.1  458.27    6033  457.51  6041.2  458.17  6077.7  458.38
  6127.5  457.99  6416.1  462.78    6471   463.2  6879.2  472.22  6936.4  472.52
#Mann= 7 ,-1 , 0
  4116.4     .08       0  4154.7     .16       0  4427.1     .05       0
  4443.9    .033       0  4449.9     .05       0  5374.9     .12       0
  5582.8     .05       0
Bank Sta=4365.2,5560.9
XS Rating Curve= 0 ,0
Exp/Cntr=0.3,0.1

Type RM Length L Ch R = 1 ,37944   ,624,624,624
BEGIN DESCRIPTION:
HOLMAN CREEK 48.0
END DESCRIPTION:
XS GIS Cut Line= 4
      3543468.72     10585136.99       3542596.3     10584212.48
      3541502.55     10583830.54       3540692.1     10583591.64
#Sta/Elev= 30
  3487.8  486.59  3552.7  486.38  3623.5  483.07  3687.5  483.11  3765.1  481.11
  3927.8   474.1  4019.6  471.87  4047.9  469.88  4117.5   468.8  4175.4  467.37
  4189.5  467.93  4196.4  466.72  4255.8  465.35  4348.9  461.73  4401.9  458.55
  4465.4  454.79  4472.3  455.42  4486.5  454.64  5660.7  454.53  5663.5  454.03
  5666.7  454.53  5927.2   458.4  6076.1  459.44  6181.3  462.84  6366.2  464.97
  6397.5  466.91  6595.6   474.3  6626.9   474.4    6683  476.77  6762.4   478.3
#Mann= 7 ,-1 , 0
  3487.8     .05       0  4117.5     .08       0  4255.8     .12       0
  4348.9     .05       0  5660.7    .033       0  5666.7     .05       0
    6683     .16       0
Bank Sta=4401.9,5927.2
XS Rating Curve= 0 ,0
Exp/Cntr=0.3,0.1

Type RM Length L Ch R = 1 ,37320   ,531,531,531
BEGIN DESCRIPTION:
HOLMAN CREEK 46.0
END DESCRIPTION:
XS GIS Cut Line= 4
      3543399.25     10584325.34      3542782.93     10583600.51
       3542036.4     10583396.51      3540131.65     10582806.43
#Sta/Elev= 30
  3818.4  473.55  3895.1  474.29  3925.7  473.11  3932.3  471.28  3938.3  471.16
  3960.9  467.61  4053.1  459.39    4074  457.12  4124.5  454.47  5016.5  454.42
  5019.2  453.92  5022.5  454.42  5463.7  454.69  5534.5  456.32  5582.2  457.02
  5646.2  455.97  5663.4  457.47  5757.6  458.53  6093.7  465.01    6196  467.35
  6351.7  468.07  6557.8  466.34    6815  469.86  6997.3  470.11    7339  474.53
  7359.4  476.02  7453.6  476.78  7474.6  478.69    7485  477.89  7537.8  478.86
#Mann= 9 ,-1 , 0
  3818.4     .05       0  3895.1     .08       0  3938.3     .05       0
  5016.5    .033       0  5022.5     .05       0  5534.5     .16       0
  5582.2     .05       0  6093.7     .08       0    6196     .05       0
Bank Sta=4053.1,5757.6
XS Rating Curve= 0 ,0
Exp/Cntr=0.3,0.1

Type RM Length L Ch R = 1 ,36789   ,731,731,731
BEGIN DESCRIPTION:
HOLMAN CREEK 45.0
END DESCRIPTION:
XS GIS Cut Line= 3
      3544542.12     10583791.65      3542742.11     10583041.64
       3541542.1     10581941.64
#Sta/Elev= 30
    3050  489.65  3141.4  487.06  3234.2  485.12  3246.9  483.77  3288.4  482.25
    3310  483.19  3515.9  475.27  3714.6  474.24  3894.9   468.2  4090.2  458.26
  4195.6  457.02  4263.9  457.41    4301  456.08  4406.4   461.6  4458.3  461.82
  4511.9   459.6  4617.3  454.86  4715.4  454.54  4718.1  454.04  4721.4  454.54
  5679.2  454.69  5725.7  457.49  5757.5  459.48  5822.5  462.58  5948.7  466.71
  6104.1  468.46  6342.7     474  6472.2  476.41  6528.5   478.1  6627.9  481.42
#Mann= 18 ,-1 , 0
    3050      .1       0  3141.4     .05       0  3246.9     .16       0
  3894.9     .12       0  4090.2     .05       0  4195.6      .1       0
    4301     .05       0  4406.4     .08       0  4458.3     .05       0
  4511.9     .08       0  4617.3     .05       0  4715.4    .033       0
  4721.4     .05       0  5725.7     .16       0  5822.5     .05       0
  6342.7      .1       0  6472.2     .12       0  6528.5      .1       0
Bank Sta=4511.9,5757.5
XS Rating Curve= 0 ,0
Exp/Cntr=0.3,0.1

Type RM Length L Ch R = 1 ,36058   ,1417,1417,1417
BEGIN DESCRIPTION:
HOLMAN CREEK 43.0
END DESCRIPTION:
XS GIS Cut Line= 3
      3544966.08     10582315.78      3543212.62     10582476.37
      3541598.06       10581821.
#Sta/Elev= 30
  2895.9  492.28  2990.3   489.7  3151.5  481.79  3251.2  479.67  3331.7  480.36
    3412  478.24  3477.4  478.55  3542.6  478.45  3602.8  475.09  3780.5  468.54
  3811.4  465.86  3944.2  458.85  4048.7  457.48  4054.7  457.23  4074.8  455.19
  4115.7  454.64  5317.8   454.5  5320.6     454  5323.8   454.5  5422.6  454.66
  5486.7  456.69    5511  457.61  5559.3  458.76  5801.9  464.38    5907  466.04
  6012.1  469.87  6194.5  475.85  6216.1  476.44  6340.2   480.1  6399.2  482.12
#Mann= 16 ,-1 , 0
  2895.9      .1       0  3151.5     .16       0  3251.2     .05       0
  3477.4      .1       0  3811.4     .08       0  4048.7     .05       0
  5317.8    .033       0  5323.8     .05       0  5486.7     .12       0
  5559.3     .16       0  5801.9     .12       0    5907     .05       0
  6012.1      .1       0  6194.5     .05       0  6216.1      .1       0
  6340.2     .05       0
Bank Sta=4054.7,5511
XS Rating Curve= 0 ,0
Exp/Cntr=0.3,0.1

Type RM Length L Ch R = 1 ,34641   ,29,29,29
BEGIN DESCRIPTION:
HOLMAN CREEK 42.0
END DESCRIPTION:
XS GIS Cut Line= 6
      3544166.43     10580633.49      3543628.42     10581009.83
      3543311.58     10581099.89      3542663.79     10581145.46
       3542379.5      10581367.9      3542093.09     10581465.54
#Sta/Elev= 30
  3507.9  472.06  3567.5  470.61  3618.6  459.02  3781.7  455.32  3934.4  457.11
  3964.5   460.9  3985.6  458.64  4016.2  460.03  4167.7   457.7  4295.5  458.75
  4300.7   456.4  4334.5  458.98  4379.6  456.22  4523.9   455.1  5067.9  456.52
  5121.9  455.67  5191.8  456.68  5194.3  454.81  5197.1  454.31  5200.3  454.81
  5220.2  459.52  5225.7  456.59  5235.3  458.34  5256.1  455.84    5426  460.19
  5432.9  457.68    5483   457.9  5514.6  460.39  5536.3  463.33  5813.5  466.55
#Mann= 10 ,-1 , 0
  3507.9      .1       0  3781.7     .08       0  4016.2      .1       0
  4167.7     .08       0  5067.9     .05       0  5121.9     .08       0
  5194.3     .07       0  5200.3     .08       0    5483     .16       0
  5514.6     .05       0
Bank Sta=4334.5,5220.2
XS Rating Curve= 0 ,0
Exp/Cntr=0.3,0.1

Type RM Length L Ch R = 1 ,34612   ,43,43,43
BEGIN DESCRIPTION:
HOLMAN CREEK 41.0
END DESCRIPTION:
XS GIS Cut Line= 6
      3544145.25     10580620.24      3543583.97     10580989.61
      3543308.36     10581059.05      3542727.85     10581092.69
      3542362.18     10581353.11      3542067.93     10581442.94
#Sta/Elev= 30
  3546.6  471.44  3600.1   469.6  3621.4   462.3    3644  459.11  3779.6  455.88
  3796.3  455.63  3802.3  454.86    3805  454.36  3808.3  454.86  3826.6  455.66
  3958.2  457.17  4037.6  465.59  4087.5  463.83  4102.5  463.65  4294.5   464.7
  4330.4   460.6  4335.6  464.15  4371.5  459.81  4376.6  463.27  4407.4   460.7
  4412.6  464.06  4448.5  461.67  4453.7  464.25  4540.5  464.86  5097.8   461.6
  5175.7  463.54  5193.8  461.14  5214.3  463.56  5520.4  462.48  5849.4  466.35
#Mann= 7 ,-1 , 0
  3546.6      .1       0  3779.6     .08       0  3802.3     .07       0
  3808.3     .08       0  4087.5      .1       0  4102.5     .08       0
  5520.4     .05       0
Bank Sta=3796.3,3826.6
XS Rating Curve= 0 ,0
Exp/Cntr=0.3,0.1

Type RM Length L Ch R = 1 ,34569   ,519,519,519
BEGIN DESCRIPTION:
HOLMAN CREEK 40.0
END DESCRIPTION:
XS GIS Cut Line= 6
      3544121.54     10580578.45      3543554.69     10580963.87
      3543384.55     10581021.17      3542620.66     10581088.87
      3542348.96     10581331.06      3542067.68     10581418.74
#Sta/Elev= 30
  3573.5  470.97  3632.6  469.38    3656  462.14  3683.1  458.34  3791.1     455
  3987.7  456.41  4029.8  460.88  4066.2  460.82  4175.1   459.7  4273.1  459.51
  4339.3  455.64  4378.7  454.11  4393.8  455.71    4420  453.64  4425.3  456.46
  4531.5  451.94    4952  449.82    4959  449.23  4961.7  448.73    4965  449.23
    4972  449.86  5160.2  452.91  5195.6  451.48  5200.8  453.39  5217.2  451.59
    5238  454.54  5252.6   452.8  5528.6  462.46  5691.7   462.4    5868  466.33
#Mann= 9 ,-1 , 0
  3573.5      .1       0  3791.1     .08       0  4066.2      .1       0
  4175.1     .08       0  4339.3      .1       0  4378.7     .08       0
    4959     .07       0    4965     .08       0  5528.6     .05       0
Bank Sta=4952,4972
XS Rating Curve= 0 ,0
Exp/Cntr=0.3,0.1

Type RM Length L Ch R = 1 ,34050   ,213,213,213
BEGIN DESCRIPTION:
HOLMAN CREEK 38.01
END DESCRIPTION:
XS GIS Cut Line= 2
        3544136.     10580459.02      3541629.03      10580674.3
#Sta/Elev= 30
  3676.4  470.04  3765.6  468.67  3891.1  464.38  3971.4  457.39  4116.5  453.58
  4157.9   450.6  4573.6  439.15  4764.3  437.49  4904.8  439.17  4914.8  439.01
  4932.1  435.33  4937.1  435.42    4955  439.76    4965  438.99  4985.1   435.4
  5002.2  429.82  5004.9  429.32  5008.2  429.82  5025.2  438.49    5226  437.87
  5412.7  441.42  5520.4  444.17  5657.6  443.45  5677.6  447.21  5697.7  448.64
  5978.7  450.42    6049  457.19  6098.6  458.81  6103.7   457.9  6192.6  458.86
#Mann= 5 ,-1 , 0
  3676.4      .1       0  4157.9     .16       0  5002.2     .07       0
  5008.2     .16       0  5412.7     .05       0
Bank Sta=4965,5025.2
XS Rating Curve= 0 ,0
Exp/Cntr=0.3,0.1

Type RM Length L Ch R = 1 ,33837   ,26,26,26
BEGIN DESCRIPTION:
HOLMAN CREEK 39.01
END DESCRIPTION:
XS GIS Cut Line= 4
      3544297.56     10580166.52      3542805.96     10580344.47
      3542723.49     10580394.39      3541525.22     10580535.23
#Sta/Elev= 30
  3442.3  469.09  3518.3  465.92  3535.4  466.46  3595.4  464.66  3695.5  460.11
  3953.1   452.9  3991.6  449.85  4062.1  448.65  4118.1  445.06  4237.7  442.89
  4337.7   442.1  4460.8  441.38  4793.9  438.36  4938.3   438.1  4988.6  436.52
  4995.7   431.6  5001.1  430.32  5003.8  429.82  5007.1  430.32  5025.4  438.12
  5132.9  436.09    5440   439.5  5553.5   441.2  5610.2  442.45  5653.6  444.32
  5787.4  448.88  5898.1  448.07  5958.5  450.86  5998.1  457.17  6247.4  462.54
#Mann= 13 ,-1 , 0
  3442.3     .05       0  3535.4      .1       0  3595.4     .16       0
  4237.7      .1       0  4337.7     .16       0  4460.8     .12       0
  4793.9     .16       0  5001.1     .07       0  5007.1     .16       0
    5440     .12       0  5553.5     .16       0  5610.2     .12       0
  5653.6     .05       0
Bank Sta=4988.6,5025.4
XS Rating Curve= 0 ,0
Exp/Cntr=0.3,0.1

Type RM Length L Ch R = 1 ,33811   ,146,146,146
BEGIN DESCRIPTION:
HOLMAN CREEK 39.0
END DESCRIPTION:
XS GIS Cut Line= 4
      3544296.48     10580146.34      3542788.02     10580327.76
      3542704.69     10580372.03      3541498.97     10580517.87
#Sta/Elev= 30
  3430.1  468.73  3522.5   465.3  3539.8  465.07  3797.1  457.14  3846.9  452.78
  4119.4  444.92  4223.7  445.02  4323.8  445.13  4381.3  442.59  4504.5  444.25
  4606.5  440.72  4688.6  442.83    4804  439.98  4925.2  441.68  4970.7  436.79
  4989.7  429.87  4992.5  429.37  4995.7  429.87  5014.7  436.23  5036.7  437.86
  5066.5  432.59  5086.9  436.26    5127  437.08  5410.3  439.51  5536.8  441.04
    5737  446.47  5829.4  449.89  5911.3   448.6  5983.2  457.39  6258.3  463.17
#Mann= 12 ,-1 , 0
  3430.1     .05       0  3522.5      .1       0  3539.8     .16       0
  4223.7      .1       0  4323.8     .16       0  4504.5     .12       0
    4804     .16       0  4989.7     .07       0  4995.7     .16       0
  5410.3     .12       0  5536.8     .16       0    5737     .05       0
Bank Sta=4970.7,5014.7
XS Rating Curve= 0 ,0
Exp/Cntr=0.3,0.1

Type RM Length L Ch R = 1 ,33665   ,75,75,75
BEGIN DESCRIPTION:
HOLMAN CREEK 39.02
END DESCRIPTION:
XS GIS Cut Line= 4
       3544249.1     10580049.33       3542745.2     10580203.59
       3542578.1     10580275.21      3541527.97     10580426.77
#Sta/Elev= 30
  3376.2   464.7  3417.2   463.5  3735.1  449.69  3983.7   446.9  4016.2  446.32
  4095.8  445.54  4215.8  444.57  4315.7  443.64  4754.8  438.97  4891.9  437.78
  4919.8  434.76    4967  437.35    4993  429.68  4995.7  429.18    4999  429.68
    5025  437.49  5080.4  440.35    5245  439.53  5356.8  438.27  5361.8   440.9
  5427.1  439.84  5432.2  442.22  5497.5  440.38  5502.5  443.31  5687.7   446.4
  5924.7  453.69  5975.1   458.6    5990  456.37  6045.8  461.99  6130.8  462.71
#Mann= 13 ,-1 , 0
  3376.2     .05       0  3417.2     .16       0  3983.7      .1       0
  4016.2     .05       0  4095.8     .16       0  4215.8      .1       0
  4315.7     .12       0  4754.8     .16       0    4993     .07       0
    4999     .16       0    5245     .12       0  5432.2     .16       0
  5687.7     .05       0
Bank Sta=4967,5025
XS Rating Curve= 0 ,0
Exp/Cntr=0.3,0.1

Type RM Length L Ch R = 1 ,33590   ,985,985,985
BEGIN DESCRIPTION:
HOLMAN CREEK 39.03
END DESCRIPTION:
XS GIS Cut Line= 4
      3544433.57      10579999.6      3542638.86     10580179.72
      3542521.67     10580264.36      3541512.55      10580392.4
#Sta/Elev= 30
  3114.4  467.66  3549.9  455.44  3628.4   449.8  3769.1  452.29  3812.2  448.88
  3938.3  449.74  3990.6   446.8  4038.1  449.28  4070.6   448.4  4085.9  453.45
  4137.9  452.54    4255  452.67  4442.5  446.61  4492.8  441.38  4661.1  439.19
  4975.4  436.65  4981.6  430.75  4993.3  428.85    4996  428.35  4999.3  428.85
    5011  430.18  5017.2  435.37  5031.9  432.66    5038  437.13  5052.7  437.84
    5168  436.66  5366.4  437.68  5605.1  444.22  5777.9  456.37  6079.9   464.2
#Mann= 13 ,-1 , 0
  3114.4     .05       0  3549.9     .16       0  3812.2      .1       0
  3938.3     .05       0  4038.1      .1       0  4137.9     .05       0
    4255     .12       0  4661.1     .16       0  4993.3     .07       0
  4999.3     .16       0    5168     .12       0  5366.4     .16       0
  5605.1     .05       0
Bank Sta=4975.4,5017.2
XS Rating Curve= 0 ,0
Exp/Cntr=0.3,0.1

Type RM Length L Ch R = 1 ,32605   ,830,830,830
BEGIN DESCRIPTION:
HOLMAN CREEK 38.0
END DESCRIPTION:
XS GIS Cut Line= 3
      3543642.86     10579845.32      3543382.48     10579940.79
      3541795.52     10579515.87
#Sta/Elev= 30
  3825.9  463.35  4003.2  458.46    4114  457.61  4265.9  452.46  4372.8  450.18
  4485.7  444.78  4544.1  442.35  4671.2  440.57  4772.5  438.64  4891.9  435.65
  4921.5  436.24  4955.4  435.27  4974.1  434.54  4990.9  428.61  4993.7  428.11
  4996.9  428.61  5003.8  428.62  5014.6  433.59    5025  435.54  5123.9  434.65
  5202.6  436.53  5265.3  440.57  5357.6  444.82  5433.8  445.33  5490.8  444.21
  5623.7  446.11  5697.9   449.9  5713.2  453.22  5728.9  455.04  5746.1  453.46
#Mann= 13 ,-1 , 0
  3825.9     .05       0  4265.9     .16       0  4485.7     .05       0
  4671.2     .16       0  4772.5     .12       0  4891.9     .16       0
  4955.4     .12       0  4990.9     .07       0  4996.9     .12       0
  5202.6     .07       0  5265.3     .12       0  5357.6     .05       0
  5713.2     .08       0
Bank Sta=4974.1,5025
XS Rating Curve= 0 ,0
Exp/Cntr=0.3,0.1

Type RM Length L Ch R = 1 ,31775   ,933,933,933
BEGIN DESCRIPTION:
HOLMAN CREEK 36.0
END DESCRIPTION:
XS GIS Cut Line= 3
      3544184.87     10578917.35      3542848.03     10578926.03
      3542019.08     10579021.51
#Sta/Elev= 30
  3469.5  476.69  3642.3  476.64  3823.8  469.72  3952.3  463.24  4012.3  459.03
  4315.2  446.74  4352.3  444.32  4372.3  444.55  4472.8  441.12  4489.4  440.69
  4542.3  438.11  4622.3  437.33  4687.3  435.27  4772.3  433.66  4953.3  434.45
  4987.5  433.56  4993.5   430.4  5000.6  430.25  5003.3  429.75  5006.6  430.25
  5023.7  434.25  5033.8  434.91    5086  434.32  5124.4   433.6  5186.1  433.87
  5249.5  434.89  5315.6   438.2  5466.6  448.83  5537.1  451.14  5640.8  450.94
#Mann= 11 ,-1 , 0
  3469.5     .05       0  3823.8     .16       0  4315.2     .12       0
  4472.8     .16       0  4489.4     .07       0  4687.3     .12       0
  5000.6     .07       0  5006.6     .12       0    5086     .16       0
  5186.1     .07       0  5315.6     .05       0
Bank Sta=4987.5,5023.7
XS Rating Curve= 0 ,0
Exp/Cntr=0.3,0.1

Type RM Length L Ch R = 1 ,30842   ,18,18,18
BEGIN DESCRIPTION:
HOLMAN CREEK 34.03
END DESCRIPTION:
XS GIS Cut Line= 5
       3543124.9     10578275.09       3542111.9     10578246.44
      3541864.51     10578230.82      3541781.18     10578202.17
      3541076.23     10578187.86
#Sta/Elev= 30
    4139  449.43    4185  448.49  4257.9  447.02  4442.3  442.42    4542  437.41
    4712  432.61  4852.1  433.18  4972.1   432.1  4982.1  430.68  4989.1   426.5
  4991.9     426  4995.1   426.5  5002.1  427.14  5012.1  431.75  5022.1  432.96
  5102.2  440.59  5141.2  442.92    5254  438.86  5332.6  437.29  5352.6  437.76
  5459.6  435.56  5490.4  434.76  5527.5  436.04  5627.5  437.02  5837.5  443.11
  5856.2  444.25  5877.6  446.04  5927.6  447.62  6037.6  448.62  6193.5  453.88
#Mann= 8 ,-1 , 0
    4139     .05       0    4185     .08       0  4257.9     .05       0
  4989.1     .04       0  4995.1     .05       0    5254     .08       0
  5459.6     .05       0  5856.2     .08       0
#XS Ineff= 2 , 0
                         5159.09          442.87
Permanent Ineff=
       F       F
Bank Sta=4972.1,5022.1
XS Rating Curve= 0 ,0
Exp/Cntr=0.3,0.1

Type RM Length L Ch R = 1 ,30824   ,97,97,97
BEGIN DESCRIPTION:
HOLMAN CREEK 34.0
END DESCRIPTION:
XS GIS Cut Line= 5
      3543122.71     10578257.72      3542109.73     10578229.08
      3541862.34     10578213.45      3541779.01     10578184.81
      3541075.24     10578170.53
#Sta/Elev= 30
  4137.6  449.68  4173.9  448.83  4260.4  446.97  4438.3  442.31  4526.5  438.35
  4698.4  433.26  4918.5   433.3  4938.5  431.45  4978.5  430.94  4995.5   426.7
  4998.3   426.2  5001.5   426.7  5018.6  432.69  5088.6  439.66  5138.6  442.46
  5238.3  438.86  5318.9  437.13  5346.1  437.56  5417.4  435.26  5422.7  434.14
  5448.6  435.25  5455.2  434.39  5513.9  436.53  5583.9  436.43  5654.2  437.89
  5753.6  440.44  5851.9  444.33  5889.2  446.43  5894.2  444.84  6190.9  454.07
#Mann= 10 ,-1 , 0
  4137.6     .05       0  4173.9     .08       0  4260.4     .05       0
  4995.5     .04       0  5001.5     .05       0  5238.3     .08       0
  5455.2     .05       0  5654.2     .08       0  5753.6     .05       0
  5851.9     .08       0
#XS Ineff= 2 , 0
                         5147.73          442.61
Permanent Ineff=
       F       F
Bank Sta=4978.5,5018.6
XS Rating Curve= 0 ,0
Exp/Cntr=0.3,0.1

Type RM Length L Ch R = 1 ,30727   ,16,16,16
BEGIN DESCRIPTION:
HOLMAN CREEK 34.01
END DESCRIPTION:
XS GIS Cut Line= 3
      3543227.66      10578154.9       3542136.1     10578137.54
      3541107.49     10578076.77
#Sta/Elev= 30
  4056.7  452.41  4187.8  452.45  4286.7  450.54  4422.3  446.72  4583.3  438.52
  4632.3  435.59  4802.3  432.88  4903.6   432.9    4914  432.63  4972.4  431.85
  4989.4  426.45  4992.1  425.95  4995.4  426.45  5002.4  427.24  5022.4  432.71
  5132.4  437.78  5165.5  438.43    5197  436.72  5272.6   434.7  5382.8  435.38
  5412.8  431.15  5432.9  435.36    5473  436.21    5513  435.82  5563.1   437.5
  5670.7  438.71  5793.5  442.54  5913.7   443.3  5953.8  446.72  6178.8  452.96
#Mann= 11 ,-1 , 0
  4056.7     .08       0  4187.8     .05       0  4286.7     .08       0
  4583.3     .05       0  4903.6     .16       0    4914     .05       0
  4989.4     .04       0  4995.4     .05       0    5197     .08       0
    5473     .05       0  5670.7     .08       0
#XS Ineff= 2 , 0
                         5166.19          438.48
Permanent Ineff=
       F       F
Bank Sta=4972.4,5022.4
XS Rating Curve= 0 ,0
Exp/Cntr=0.3,0.1

Type RM Length L Ch R = 1 ,30711   ,339,339,339
BEGIN DESCRIPTION:
HOLMAN CREEK 34.02
END DESCRIPTION:
XS GIS Cut Line= 3
      3543227.69     10578139.71       3542136.1     10578122.34
      3541107.42     10578061.58
#Sta/Elev= 30
  4063.1  452.92  4158.6  452.81  4338.7  450.53  4457.1  446.48  4538.7  442.47
  4589.1  438.84  4638.8  436.02  4688.8  434.56    4901  432.15  4950.5  432.21
  4958.8  432.04  4978.8  429.92  4985.8  426.77  4988.5  426.27  4991.8  426.77
  4998.8  427.27  5018.8   432.8  5128.8  437.95  5192.8  436.89    5259  434.02
  5389.2   434.8  5409.3  431.38  5429.3  434.76  5478.8  435.85  5676.5   438.3
  5870.1  443.52  5920.2  442.94  5950.2  447.13  5993.7  447.52  6185.3   453.2
#Mann= 12 ,-1 , 0
  4063.1     .08       0  4158.6     .16       0  4457.1     .08       0
  4589.1     .05       0    4901     .16       0  4950.5     .05       0
  4985.8     .04       0  4991.8     .05       0  5192.8     .08       0
  5478.8     .05       0  5676.5     .08       0  5993.7     .05       0
#XS Ineff= 2 , 0
                         5159.09           438.1
Permanent Ineff=
       F       F
Bank Sta=4958.8,5018.8
XS Rating Curve= 0 ,0
Exp/Cntr=0.3,0.1

Type RM Length L Ch R = 1 ,30372   ,1159,1159,1159
BEGIN DESCRIPTION:
HOLMAN CREEK 33.0
END DESCRIPTION:
XS GIS Cut Line= 3
      3542954.92     10577789.56      3542504.95     10577839.56
      3540706.06     10577389.83
#Sta/Elev= 30
  4424.8  458.67  4518.2  458.38  4581.5  454.19  4672.1  444.43  4719.4  436.31
  4757.6  432.42    4820  430.81  4975.2     432  5001.2   426.8  5003.9   426.3
  5007.2   426.8  5011.3   429.8  5024.8  432.49  5270.6  431.07  5447.4  434.46
  5547.3  439.76  5712.2  445.96    5870  448.49  5918.4  445.74  6088.5  445.14
  6096.8  447.28  6170.9  448.31  6189.6  450.05  6230.8  448.48  6371.9  453.22
  6413.1  453.14  6531.2  458.45  6583.2  460.76  6653.1  461.31  6731.8  461.28
#Mann= 6 ,-1 , 0
  4424.8     .16       0  5001.2     .07       0  5007.2     .16       0
  5270.6     .05       0  6531.2      .1       0  6653.1     .05       0
Bank Sta=4975.2,5024.8
XS Rating Curve= 0 ,0
Exp/Cntr=0.3,0.1

Type RM Length L Ch R = 1 ,29213   ,667,667,667
BEGIN DESCRIPTION:
HOLMAN CREEK 31.0
END DESCRIPTION:
XS GIS Cut Line= 3
      3543259.49     10577467.46      3541540.76      10576651.5
        3541098.     10576599.41
#Sta/Elev= 30
  3797.7  461.01  3828.2  461.72  3845.4  460.36  3964.6  458.97  4288.3  441.96
  4356.5  443.99  4424.7  442.88  4724.7  428.04    4754   430.5  4969.6  429.38
  4998.4   423.5  5001.2     423  5004.4   423.5  5020.1  429.58  5032.2  430.97
  5127.5  429.22  5189.6  429.68  5314.5  433.86  5400.3  436.93  5503.4  439.02
  5685.2  445.88    5738  446.84  5759.3  444.75  5789.6  446.76  5870.1  448.39
  5914.2  447.67  6011.1  450.64  6102.3  451.38  6121.8  453.47  6146.1  451.61
#Mann= 8 ,-1 , 0
  3797.7     .16       0  4998.4     .07       0  5004.4     .16       0
  5020.1     .12       0  5127.5     .05       0  5314.5     .16       0
  5400.3     .05       0  6102.3      .1       0
Bank Sta=4969.6,5020.1
XS Rating Curve= 0 ,0
Exp/Cntr=0.3,0.1

Type RM Length L Ch R = 1 ,28546   ,907,907,907
BEGIN DESCRIPTION:
HOLMAN CREEK 29.0
END DESCRIPTION:
XS GIS Cut Line= 3
      3543598.89     10576907.79      3542361.92     10576378.28
      3541012.11     10576269.78
#Sta/Elev= 30
  3493.3  479.06  3642.1  476.86  3747.9  471.95  3952.9  450.33  4005.5  446.12
    4029  442.95  4058.1  442.04  4105.2  436.34    4205  431.61  4263.1  431.72
  4349.1   428.2    4450  427.38  4585.1  428.21  4685.7  426.93  4767.3  428.45
  4979.1  428.41  4996.2   422.8  4998.9   422.3  5002.2   422.8  5019.2   428.3
  5101.2  430.45  5320.2  443.68  5361.9  444.54  5479.5  442.43  5612.1  444.19
  5641.2  443.47  5801.7  447.94  5971.7  450.16  6158.4  453.59    6193  454.65
#Mann= 8 ,-1 , 0
  3493.3     .16       0    4450     .12       0  4585.1     .16       0
  4996.2     .07       0  5002.2     .16       0  5101.2     .05       0
  5971.7      .1       0  6158.4     .05       0
Bank Sta=4979.1,5019.2
XS Rating Curve= 0 ,0
Exp/Cntr=0.3,0.1

Type RM Length L Ch R = 1 ,27639   ,622,622,622
BEGIN DESCRIPTION:
HOLMAN CREEK 27.0
END DESCRIPTION:
XS GIS Cut Line= 4
      3544054.66     10576842.71      3542934.84     10576000.68
        3542414.     10575909.53      3541576.75     10575740.35
#Sta/Elev= 30
  3481.8  477.18    3576  474.68  3726.9  470.84    3956  471.51  4155.9  468.02
  4320.4   458.1  4659.6   426.7  4926.3  426.73    4977  428.12  4994.3  423.02
  4997.1  422.52  5000.3  423.02  5017.4  426.98  5027.8  427.91  5068.4  426.93
  5132.7  430.06  5195.8  432.34  5342.5  433.53  5478.3  438.84  5568.8  444.27
  5617.6  445.26    5740  443.42  5903.3  444.39  5944.1  443.28  6046.1  446.39
  6056.3   443.6  6066.5  445.26  6107.3  445.44  6199.1  443.49  6265.8  446.97
#Mann= 7 ,-1 , 0
  3481.8     .12       0    3576     .16       0  4659.6     .12       0
  4994.3     .07       0  5000.3     .12       0  5132.7     .05       0
  5568.8     .16       0
Bank Sta=4977,5017.4
XS Rating Curve= 0 ,0
Exp/Cntr=0.3,0.1

Type RM Length L Ch R = 1 ,27017   ,738,738,738
BEGIN DESCRIPTION:
HOLMAN CREEK 25.0
END DESCRIPTION:
XS GIS Cut Line= 4
      3544306.34     10576456.39      3543225.64     10575514.57
      3542448.73     10575241.13      3541389.67     10575136.96
#Sta/Elev= 30
  3358.7  472.92  3712.1  457.85  3875.4  448.01  4038.7  440.74  4307.4  434.08
  4470.7  425.47  4611.8  424.34  4683.3  423.55  4821.6  425.26  4976.2  425.82
  4991.4  422.42  4994.2  421.92  4997.4  422.42  5018.6  426.05  5061.7  425.48
  5260.3  429.43  5360.7  432.05    5436  432.15  5495.6  431.19  5559.2  428.19
  5716.4  430.22  5749.6  431.52  5963.6  440.37  6305.8  445.95  6424.8  446.37
  6466.5  447.01  6475.3  445.95  6546.9  445.49  6576.6  447.92    6680  448.29
#Mann= 10 ,-1 , 0
  3358.7     .16       0  4611.8     .12       0  4821.6     .16       0
  4991.4     .07       0  4997.4     .16       0  5260.3     .05       0
    5436     .16       0  5716.4     .05       0  5749.6     .16       0
  6424.8     .05       0
Bank Sta=4976.2,5018.6
XS Rating Curve= 0 ,0
Exp/Cntr=0.3,0.1
