--- WHITE ROCK CREEK.prj (project) ---

Proj Title=WHITE ROCK CREEK Base Level Engineering
Current Plan=p01
Default Exp/Contr=0.3,0.1
English Units
Geom File=g01
Flow File=f01
Plan File=p01
BEGIN DESCRIPTION:
WHITE ROCK CREEK
END DESCRIPTION:

--- WHITE ROCK CREEK.p01 (plan) ---

Plan Title=Multiple Run
Short Identifier=Multiple
Geom File=g01
Flow File=f01
Subcritical Flow
K Sum by GR= 0
Std Step Tol= 0.01
Critical Tol= 0.01
Num of Std Step Trials= 20
Max Error Tol= 0.3
Flow Tol Ratio= 0.001
Split Flow NTrial= 30
Split Flow Tol= 0.02
Split Flow Ratio= 0.02
Log Output Level= 0
Friction Slope Method= 1
Unsteady Friction Slope Method= 2
Unsteady Bridges Friction Slope Method= 1
Parabolic Critical Depth
Global Vel Dist=  1 , 1 , 1
Global Log Level= 0
CheckData=True
Encroach Param= -1, 0, 0, 0
BEGIN DESCRIPTION:
Multiple Run
END DESCRIPTION:

--- WHITE ROCK CREEK.f01 (steady flow) ---

Flow Title=Multiple
Number of Profiles=7
Profile Names=10-year,25-year,50-year,1pct_min,100-year,1pct_plu,500-year
River Rch & RM= WHITE ROCK CREEK,Reach-1,27875
     751     999    1197    1046    1414    1913    1968
River Rch & RM= WHITE ROCK CREEK,Reach-1,23096
    1732    2422    2998    2702    3653    4941    5412
River Rch & RM= WHITE ROCK CREEK,Reach-1,17570
    2434    3465    4344    3959    5354    7240    8116
River Rch & RM= WHITE ROCK CREEK,Reach-1,17116
    2734    3886    4864    4422    5980    8088    9023
River Rch & RM= WHITE ROCK CREEK,Reach-1,6783
    2787    3965    4965    4517    6109    8262    9228
River Rch & RM= WHITE ROCK CREEK,Reach-1,4489
    3286    4704    5915    5401    7304    9878   11114
Boundary for River Rch & Prof#=WHITE ROCK CREEK,Reach-1,1
Up Type=0
Dn Type=3
Dn Slope=0.005
Boundary for River Rch & Prof#=WHITE ROCK CREEK,Reach-1,2
Up Type=0
Dn Type=3
Dn Slope=0.005
Boundary for River Rch & Prof#=WHITE ROCK CREEK,Reach-1,3
Up Type=0
Dn Type=3
Dn Slope=0.005
Boundary for River Rch & Prof#=WHITE ROCK CREEK,Reach-1,4
Up Type=0
Dn Type=3
Dn Slope=0.005
Boundary for River Rch & Prof#=WHITE ROCK CREEK,Reach-1,5
Up Type=0
Dn Type=3
Dn Slope=0.005
Boundary for River Rch & Prof#=WHITE ROCK CREEK,Reach-1,6
Up Type=0
Dn Type=3
Dn Slope=0.005
Boundary for River Rch & Prof#=WHITE ROCK CREEK,Reach-1,7
Up Type=0
Dn Type=3
Dn Slope=0.005

--- WHITE ROCK CREEK.g01 (geometry) ---

Geom Title=Existing Conditions

River Reach=WHITE ROCK CREEK,Reach-1
Reach XY= 30
      3549845.80     10586841.51      3549998.29     10586548.91
      3549787.31     10585826.53      3550485.53     10585336.97
      3550571.36     10584296.87      3551271.88     10583118.05
      3550683.59     10581154.23      3549257.37     10579560.48
      3548755.83     10578014.50      3548417.38     10577753.98
      3548398.84     10577042.99      3548177.95     10576639.57
      3547692.34     10576346.60      3547652.11     10574641.68
      3548241.48     10573411.18      3548145.75     10572748.18
      3547808.29     10572447.62      3547945.01     10572339.11
      3547723.77     10572155.53      3547674.21     10571565.36
      3547083.12     10571066.98      3547291.45     10570641.45
      3546833.62     10569765.86      3546700.14     10568187.61
      3545822.39     10566707.40      3545815.40     10566163.09
      3546117.00     10566103.92      3546064.36     10565537.12
      3546330.39     10565196.06      3546281.51     10564426.40

Type RM Length L Ch R = 1,27875,837,837,837
BEGIN DESCRIPTION:
WHITE ROCK CREEK 47.0
END DESCRIPTION:
XS GIS Cut Line= 4
      3550787.35     10586655.20      3550075.52     10586772.40
      3549641.49     10586772.40      3549103.30     10587024.13
#Sta/Elev= 30
  4106.2  487.00  4171.9  485.20  4233.1  484.46  4238.2  485.12  4299.4  482.98
  4304.4  483.72  4324.3  482.21  4344.6  478.55  4360.6  477.83  4395.3  482.45
  4506.8  484.46  4605.3  482.46  4881.0  480.06  4951.0  478.82  4971.0  477.87
  4981.0  476.13  4998.0  471.08  5000.8  470.58  5004.0  471.08  5011.0  473.92
  5031.0  473.95  5061.0  476.96  5089.1  478.79  5161.0  480.61  5221.0  480.18
  5390.4  481.08  5459.2  480.65  5757.8  481.33  5828.3  483.01  5855.8  483.49
#Mann=7,-1,0
  4106.2    0.08       0  4998.0    0.07       0  5004.0    0.08       0
  5089.1    0.05       0  5390.4    0.08       0  5459.2    0.05       0
  5828.3    0.08       0
Bank Sta=4998,5004
Exp/Cntr=0.3,0.1

Type RM Length L Ch R = 1,27038,1139,1139,1139
BEGIN DESCRIPTION:
WHITE ROCK CREEK 46.0
END DESCRIPTION:
XS GIS Cut Line= 4
      3551138.90     10586272.46      3550006.07     10586042.42
      3549532.98     10586124.89      3548475.53     10585851.86
#Sta/Elev= 30
  3698.8  494.66  4054.5  485.06  4195.5  482.96  4246.5  480.32  4552.7  475.14
  4580.2  469.85  4585.3  471.52  4593.5  469.19  4603.7  468.61  4624.1  468.88
  4644.5  472.81  4681.5  474.44  4746.5  475.92  4889.2  475.99  4950.1  474.87
  4960.3  473.98  4980.6  469.44  4997.9  467.91  5000.6  467.41  5003.9  467.91
  5031.3  471.42  5061.8  471.53  5114.9  468.25  5153.1  470.35  5169.4  472.67
  5223.9  474.54  5486.3  480.65  5603.6  480.46  6010.2  485.04  6427.1  493.31
#Mann=5,-1,0
  3698.8    0.05       0  4054.5    0.16       0  4997.9    0.07       0
  5003.9    0.16       0  5486.3    0.05       0
Bank Sta=4997.9,5003.9
Exp/Cntr=0.3,0.1

Type RM Length L Ch R = 1,25899,741,741,741
BEGIN DESCRIPTION:
WHITE ROCK CREEK 44.0
END DESCRIPTION:
XS GIS Cut Line= 4
      3551525.19     10586016.40      3550561.62     10585508.57
      3550127.59     10585274.19      3549650.16     10585013.78
#Sta/Elev= 30
  3755.4  493.94  3781.7  494.46  3804.1  493.46  3994.0  491.03  4001.5  490.91
  4154.5  488.03  4189.0  486.36  4233.6  486.26  4420.0  481.21  4425.8  480.31
  4436.3  480.91  4628.9  475.56  4753.6  471.23  4863.4  469.76  4889.8  469.08
  4914.9  467.68  4999.9  467.70  5045.6  467.52  5048.4  467.02  5051.6  467.52
  5173.6  472.76  5291.8  475.90  5482.7  476.07  5542.5  476.84  5558.7  478.14
  5564.4  477.25  5598.2  477.68  5608.0  477.28  5651.7  479.11  5881.7  483.06
#Mann=9,-1,0
  3755.4    0.16       0  3994.0    0.05       0  4001.5    0.16       0
  4863.4    0.12       0  4889.8    0.16       0  4999.9    0.12       0
  5045.6    0.07       0  5051.6    0.12       0  5598.2    0.16       0
Bank Sta=5045.6,5051.6
Exp/Cntr=0.3,0.1

Type RM Length L Ch R = 1,25158,529,529,529
BEGIN DESCRIPTION:
WHITE ROCK CREEK 42.0
END DESCRIPTION:
XS GIS Cut Line= 4
      3551559.85     10584874.88      3550761.27     10584740.34
      3550179.68     10584701.28      3549746.35     10584467.28
#Sta/Elev= 30
  4009.0  485.98  4016.9  486.47  4121.1  484.48  4458.2  475.81  4484.2  475.49
  4534.0  473.34  4554.3  473.28  4600.1  471.50  4696.3  469.13  4726.7  467.65
  4784.6  467.44  4787.3  466.94  4790.6  467.44  4816.9  467.65  4985.7  467.60
  5127.6  467.88  5158.8  468.06  5205.3  469.32  5317.9  471.75  5339.2  471.55
  5359.2  472.47  5408.1  473.20  5435.6  472.94  5457.5  473.93  5592.2  475.90
  5649.0  477.52  5665.0  477.30  5752.6  479.40  5785.0  478.69  5894.2  480.48
#Mann=8,-1,0
  4009.0    0.05       0  4458.2    0.16       0  4784.6    0.07       0
  4790.6    0.16       0  4816.9    0.05       0  4985.7    0.16       0
  5127.6    0.12       0  5205.3    0.16       0
Bank Sta=4784.6,4790.6
Exp/Cntr=0.3,0.1

Type RM Length L Ch R = 1,24629,646,646,646
BEGIN DESCRIPTION:
WHITE ROCK CREEK 41.1
END DESCRIPTION:
XS GIS Cut Line= 3
      3551503.49     10584805.46      3550489.19     10584126.97
      3550301.20     10583820.20
#Sta/Elev= 30
  3941.5  485.94  4052.4  484.05  4082.4  482.71  4103.4  482.62  4154.5  480.26
  4388.2  474.19  4571.8  469.82  4673.9  469.49  4746.0  467.62  4768.0  467.75
  5073.3  467.43  5076.0  466.93  5079.3  467.43  5086.7  467.48  5184.5  472.21
  5237.5  474.20  5243.3  475.56  5295.5  475.98  5301.4  477.41  5308.8  477.79
  5316.8  477.62  5322.7  474.73  5332.2  475.48  5338.1  473.57  5344.0  473.60
  5359.4  474.70  5367.4  478.92  5374.8  480.69  5518.7  484.94  5521.6  484.94
#Mann=8,-1,0
  3941.5    0.05       0  4388.2    0.16       0  4768.0    0.05       0
  5073.3   0.033       0  5079.3    0.05       0  5086.7    0.12       0
  5184.5    0.08       0  5518.7    0.05       0
Bank Sta=5073.3,5079.3
Exp/Cntr=0.3,0.1

Type RM Length L Ch R = 1,23983,887,887,887
BEGIN DESCRIPTION:
WHITE ROCK CREEK 39.0
END DESCRIPTION:
XS GIS Cut Line= 2
      3551814.94     10584333.80      3550635.74     10583411.25
#Sta/Elev= 30
  3918.9  477.67  4043.6  477.92  4143.1  476.79  4187.7  476.83  4236.2  476.38
  4242.6  475.86  4250.7  476.60  4286.0  475.06  4321.2  475.01  4385.4  473.21
  4443.4  472.33  4670.9  467.51  4738.7  467.46  4741.5  466.96  4744.7  467.46
  5098.0  468.72  5126.9  468.24  5133.3  467.59  5147.7  468.02  5232.7  473.09
  5255.3  475.38  5261.7  475.23  5305.0  479.05  5333.7  479.73  5354.8  480.28
  5361.1  479.73  5375.6  479.53  5390.1  480.59  5410.9  480.33  5416.1  480.98
#Mann=8,-1,0
  3918.9    0.05       0  4187.7    0.12       0  4443.4    0.16       0
  4670.9    0.05       0  4738.7   0.033       0  4744.7    0.05       0
  5333.7    0.08       0  5361.1     0.1       0
Bank Sta=4738.7,4744.7
Exp/Cntr=0.3,0.1

Type RM Length L Ch R = 1,23096,674,674,674
BEGIN DESCRIPTION:
WHITE ROCK CREEK 39.1
END DESCRIPTION:
XS GIS Cut Line= 2
      3552111.58     10582372.40      3550647.98     10583164.09
#Sta/Elev= 30
  3918.1  476.60  3985.1  474.64  4016.6  472.79  4065.3  471.57  4094.4  470.27
  4100.1  470.45  4110.6  468.86  4128.4  468.56  4138.2  469.40  4160.1  468.74
  4173.3  467.31  4176.0  466.81  4179.3  467.31  4315.4  467.94  4476.9  467.80
  4498.8  468.94  5327.3  467.51  5339.8  467.51  5356.0  468.27  5361.7  467.87
  5377.9  469.05  5394.1  467.52  5399.7  468.31  5443.5  469.21  5481.6  470.76
  5497.8  470.70  5509.2  471.51  5541.5  472.36  5547.2  473.00  5582.1  473.26
#Mann=6,-1,0
  3918.1    0.05       0  4016.6    0.16       0  4128.4    0.05       0
  4173.3   0.033       0  4179.3    0.05       0  5361.7     0.1       0
Bank Sta=4173.3,4179.3
Exp/Cntr=0.3,0.1

Type RM Length L Ch R = 1,22422,11,11,11
BEGIN DESCRIPTION:
WHITE ROCK CREEK 38.3
END DESCRIPTION:
XS GIS Cut Line= 6
      3551835.04     10582149.92      3551434.01     10582212.42
      3551096.33     10582224.57      3550730.02     10582264.50
      3550696.16     10582299.23      3550559.46     10583256.70
#Sta/Elev= 30
  4233.2  474.91  4357.6  473.28  4560.0  467.44  4590.4  467.92  4610.6  471.63
  4630.9  467.82  4712.0  467.89  4811.1  469.71  4865.2  469.00  4891.1  470.54
  4931.2  469.72  4991.2  472.59  5071.8  472.67  5112.0  469.03  5162.3  471.18
  5202.5  468.49  5270.4  469.55  5275.4  467.75  5345.5  468.69  5349.0  467.49
  5378.7  467.50  5479.2  467.70  5560.3  468.39  5797.0  467.20  5799.8  466.70
  5803.0  467.20  5850.5  468.41  5907.9  467.73  6250.5  472.66  6361.4  475.49
#Mann=10,-1,0
  4233.2    0.08       0  4712.0    0.05       0  4865.2    0.08       0
  5378.7    0.05       0  5479.2    0.08       0  5560.3    0.05       0
  5797.0    0.07       0  5803.0    0.05       0  5907.9    0.08       0
  6250.5    0.05       0
Bank Sta=5797,5803
Exp/Cntr=0.3,0.1

Type RM Length L Ch R = 1,22411,24,24,24
BEGIN DESCRIPTION:
WHITE ROCK CREEK 38.1
END DESCRIPTION:
XS GIS Cut Line= 6
      3551828.85     10582134.56      3551447.31     10582189.25
      3551037.16     10582217.90      3550725.96     10582249.15
      3550686.90     10582263.47      3550579.87     10582944.45
#Sta/Elev= 30
  4237.3  475.66  4554.3  467.36  4557.0  466.86  4560.3  467.36  4587.6  467.77
  4603.5  472.40  4617.8  473.41  4744.4  473.27  4788.1  473.38  4867.9  473.53
  4873.0  470.62  4998.9  473.88  5117.9  473.79  5122.9  471.94  5218.2  473.90
  5223.2  471.19  5310.3  473.32  5323.5  470.60  5380.4  473.28  5406.7  473.21
  5446.7  468.57  5451.8  473.06  5467.4  472.81  5514.3  468.13  5519.4  473.27
  5553.1  472.23  5576.9  470.81  5590.6  473.47  5713.9  473.45  6077.6  472.13
#Mann=9,-1,0
  4237.3    0.08       0  4554.3    0.07       0  4560.3    0.08       0
  4744.4    0.05       0  4788.1    0.08       0  5380.4    0.05       0
  5553.1    0.08       0  5590.6    0.05       0  5713.9    0.08       0
Bank Sta=4554.3,4560.3
Exp/Cntr=0.3,0.1

Type RM Length L Ch R = 1,22387,191,191,191
BEGIN DESCRIPTION:
WHITE ROCK CREEK 38.2
END DESCRIPTION:
XS GIS Cut Line= 6
      3551827.21     10582113.74      3551421.29     10582167.13
      3550992.82     10582197.69      3550689.34     10582221.99
      3550648.37     10582243.52      3550566.14     10582928.19
#Sta/Elev= 30
  4234.4  474.36  4560.3  467.09  4582.5  467.54  4602.7  472.19  4639.0  467.21
  4641.9  469.66  4645.9  469.66  4772.9  464.02  4777.9  468.24  4913.4  462.88
  4918.4  469.35  5050.9  460.88  5053.6  460.38  5056.9  460.88  5058.9  467.46
  5182.5  461.13  5187.5  466.96  5310.3  461.10  5315.3  465.69  5377.8  463.72
  5384.1  464.38  5389.3  467.75  5419.2  464.30  5462.5  463.04  5756.5  466.28
  5934.4  468.87  5939.4  467.41  6021.6  470.29  6026.6  468.77  6113.7  469.84
#Mann=5,-1,0
  4234.4    0.08       0  5050.9    0.07       0  5056.9    0.08       0
  5389.3    0.05       0  5756.5    0.08       0
Bank Sta=5050.9,5056.9
Exp/Cntr=0.3,0.1

Type RM Length L Ch R = 1,22196,506,506,506
BEGIN DESCRIPTION:
WHITE ROCK CREEK 38.0
END DESCRIPTION:
XS GIS Cut Line= 4
      3552132.84     10581914.82      3551221.34     10581966.90
      3550483.50     10582114.47      3550367.05     10582226.60
#Sta/Elev= 30
  3887.8  482.80  4068.8  478.14  4259.1  474.24  4469.9  467.66  4479.5  466.92
  4529.6  466.60  4569.2  465.48  4589.7  464.82  4609.7  463.02  4639.8  462.38
  4669.8  460.69  4767.8  457.92  4853.3  456.87  4874.4  456.00  4921.5  455.47
  5072.0  455.80  5178.6  455.99  5216.9  456.21  5238.5  456.50  5296.7  455.20
  5299.5  454.70  5302.7  455.20  5320.1  455.62  5358.1  459.10  5391.5  461.03
  5478.7  463.17  5591.3  462.79  5608.9  461.94  5619.5  462.71  5714.9  462.33
#Mann=14,-1,0
  3887.8    0.05       0  4469.9    0.08       0  4569.2    0.05       0
  4767.8    0.08       0  4874.4    0.05       0  4921.5    0.08       0
  5072.0    0.05       0  5178.6    0.08       0  5216.9     0.1       0
  5296.7    0.07       0  5302.7     0.1       0  5478.7    0.08       0
  5591.3    0.05       0  5619.5    0.08       0
Bank Sta=5296.7,5302.7
Exp/Cntr=0.3,0.1

Type RM Length L Ch R = 1,21690,756,756,756
BEGIN DESCRIPTION:
WHITE ROCK CREEK 37.0
END DESCRIPTION:
XS GIS Cut Line= 4
      3552206.55     10580851.47      3550973.95     10581485.13
      3550340.27     10581719.51      3549611.24     10582217.76
#Sta/Elev= 30
  3495.9  488.75  3516.8  488.47  3602.1  481.34  3669.6  481.34  3706.5  487.87
  3811.8  476.53  3817.4  472.82  3839.6  470.00  3856.1  475.58  3861.7  473.27
  3878.3  475.90  3883.9  471.86  3916.5  476.49  3944.8  472.77  3961.4  474.22
  4322.9  462.93  4486.2  458.60  4790.0  455.04  4792.7  454.54  4796.0  455.04
  5240.5  455.70  5418.8  456.19  5694.4  459.14  5802.0  458.31  5817.0  455.99
  6008.3  462.30  6131.4  464.83  6254.5  466.19  6364.2  467.76  6440.5  465.04
#Mann=13,-1,0
  3495.9    0.05       0  3516.8    0.08       0  3706.5    0.16       0
  3916.5    0.05       0  4322.9    0.16       0  4486.2    0.05       0
  4790.0   0.033       0  4796.0    0.05       0  5240.5    0.08       0
  5418.8     0.1       0  6008.3    0.05       0  6131.4    0.16       0
  6254.5    0.05       0
Bank Sta=4790,4796
Exp/Cntr=0.3,0.1

Type RM Length L Ch R = 1,20934,882,882,882
BEGIN DESCRIPTION:
WHITE ROCK CREEK 35.0
END DESCRIPTION:
XS GIS Cut Line= 4
      3551416.64     10580178.72      3550552.94     10580821.07
      3550309.88     10581016.38      3548792.13     10581341.64
#Sta/Elev= 30
  3788.8  487.72  3836.8  485.44  3851.4  483.45  3901.5  480.65  3936.9  479.74
  3951.6  478.03  4037.1  475.27  4102.6  470.50  4172.6  466.81  4216.5  462.59
  4272.8  460.67  4302.0  457.74  4366.6  455.16  4417.6  455.75  5225.5  454.94
  5228.2  454.44  5231.5  454.94  5301.9  455.01  5419.6  455.50  5694.6  457.94
  5757.7  457.95  5796.6  456.32  5845.5  455.32  6024.4  455.91  6125.8  456.82
  6306.7  465.06  6350.8  466.14  6368.7  467.87  6408.7  468.39  6729.2  470.08
#Mann=12,-1,0
  3788.8    0.05       0  4102.6    0.08       0  4417.6    0.05       0
  5225.5   0.033       0  5231.5    0.05       0  5301.9    0.08       0
  5419.6     0.1       0  5694.6    0.05       0  5796.6    0.08       0
  6024.4     0.1       0  6306.7    0.05       0  6408.7    0.16       0
Bank Sta=5225.5,5231.5
Exp/Cntr=0.3,0.1

Type RM Length L Ch R = 1,20052,1020,1020,1020
BEGIN DESCRIPTION:
WHITE ROCK CREEK 33.0
END DESCRIPTION:
XS GIS Cut Line= 4
      3551143.25     10579809.78      3549966.43     10580170.92
      3549711.06     10580337.25      3548851.56     10580972.97
#Sta/Elev= 30
  3692.7  476.76  3892.6  471.80  3903.1  470.60  3934.5  469.98  4017.9  465.71
  4093.8  460.98  4230.0  456.19  4257.5  456.22  4279.7  455.40  4393.7  456.35
  4431.6  455.66  4842.3  455.22  4845.1  454.72  4848.3  455.22  5481.1  456.01
  5545.6  456.47  5588.1  455.67  5666.7  455.61  5674.9  455.79  5681.3  456.92
  5703.4  457.50  5737.6  458.62  5824.2  463.76  5956.9  464.22  6010.7  464.30
  6052.9  465.84  6083.6  465.99  6146.8  468.02  6238.6  468.71  6297.5  468.31
#Mann=8,-1,0
  3692.7    0.05       0  4842.3   0.033       0  4848.3    0.05       0
  5481.1    0.08       0  5588.1    0.05       0  5703.4     0.1       0
  5956.9    0.05       0  6083.6    0.16       0
Bank Sta=4842.3,4848.3
Exp/Cntr=0.3,0.1

Type RM Length L Ch R = 1,19032,28,28,28
BEGIN DESCRIPTION:
WHITE ROCK CREEK 32.0
END DESCRIPTION:
XS GIS Cut Line= 5
      3550759.91     10579279.88      3549236.46     10579466.52
      3549149.65     10579481.71      3548344.53     10579603.24
      3548272.94     10579690.01
#Sta/Elev= 30
  3439.7  459.71  3597.4  458.60  3860.6  455.09  3933.4  456.64  4069.1  455.29
  4231.9  458.77  4236.9  455.64  4253.5  455.38  4293.8  458.13  4434.9  455.55
  4481.2  458.40  4777.4  455.58  4893.3  457.74  4928.6  455.56  4974.2  458.54
  4979.6  456.52  5058.9  458.79  5136.2  456.94  5222.0  455.79  5302.9  458.89
  5562.8  455.29  5626.5  457.91  5707.4  453.50  5881.9  449.99  5884.7  449.49
  5887.9  449.99  5889.9  450.22  5905.8  451.45  5948.8  462.20  5989.4  463.26
#Mann=7,-1,0
  3439.7    0.05       0  3597.4    0.16       0  3933.4    0.05       0
  5136.2    0.08       0  5881.9   0.033       0  5887.9    0.08       0
  5889.9    0.05       0
Bank Sta=5881.9,5887.9
Exp/Cntr=0.3,0.1

Type RM Length L Ch R = 1,19004,38,38,38
BEGIN DESCRIPTION:
WHITE ROCK CREEK 31.0
END DESCRIPTION:
XS GIS Cut Line= 4
      3550760.52     10579239.28      3548607.73     10579524.00
      3548281.35     10579572.61      3548230.85     10579691.41
#Sta/Elev= 30
  3424.4  468.30  3479.4  466.59  3484.5  467.47  3598.7  466.52  3950.3  465.09
  4322.6  463.85  4773.3  460.44  5021.1  460.39  5102.9  460.19  5121.4  460.05
  5702.7  460.66  5818.2  458.37  5840.7  459.81  5874.6  460.15  5894.8  458.05
  5928.1  458.78  5933.5  456.65  5939.0  456.87  5946.6  454.55  5962.6  453.28
  5976.2  449.45  5978.9  448.95  5982.2  449.45  5986.3  450.86  5991.7  449.56
  6009.9  457.30  6015.3  456.92  6022.7  459.61  6039.0  462.26  6055.0  462.30
#Mann=9,-1,0
  3424.4    0.05       0  3598.7    0.16       0  3950.3    0.05       0
  5021.1    0.16       0  5102.9    0.05       0  5121.4    0.08       0
  5840.7    0.05       0  5976.2    0.04       0  5982.2    0.05       0
Bank Sta=5976.2,5982.2
Exp/Cntr=0.3,0.1

Type RM Length L Ch R = 1,18966,148,148,148
BEGIN DESCRIPTION:
WHITE ROCK CREEK 30.1
END DESCRIPTION:
XS GIS Cut Line= 3
      3550740.32     10579214.79      3549130.12     10579418.78
      3548307.60     10579529.46
#Sta/Elev= 30
  3428.5  458.76  3593.7  457.37  4100.5  455.37  4318.6  456.70  4473.8  449.57
  4478.8  454.46  4553.9  448.44  4558.9  452.20  4634.0  447.00  4639.0  451.44
  4714.1  444.69  4719.2  449.02  4794.2  444.05  4799.3  448.75  4874.3  443.76
  4879.4  449.32  5002.3  445.24  5031.5  443.10  5034.3  442.60  5037.5  443.10
  5039.6  448.01  5180.6  444.46  5185.7  449.74  5251.4  443.75  5263.5  447.90
  5294.6  445.79  5559.8  447.69  5665.1  457.68  5810.6  458.72  5881.5  458.79
#Mann=8,-1,0
  3428.5    0.05       0  3593.7    0.16       0  4100.5    0.05       0
  5002.3    0.16       0  5031.5    0.04       0  5037.5    0.16       0
  5294.6    0.08       0  5810.6    0.05       0
Bank Sta=5031.5,5037.5
Exp/Cntr=0.3,0.1

Type RM Length L Ch R = 1,18818,303,303,303
BEGIN DESCRIPTION:
WHITE ROCK CREEK 30.0
END DESCRIPTION:
XS GIS Cut Line= 4
      3549817.66     10579216.04      3549200.51     10579260.30
      3549039.05     10579296.76      3548585.21     10579325.29
#Sta/Elev= 30
  4291.9  453.26  4477.9  450.69  4538.1  447.08  4558.1  446.42  4576.5  444.90
  4581.6  445.01  4658.4  440.21  4698.5  439.28  4758.7  438.68  4778.7  437.52
  4799.4  438.46  4808.8  438.71  4838.9  437.77  4896.0  437.01  4898.8  436.51
  4902.0  437.01  4910.6  437.42  4919.3  438.72  4924.9  438.90  4937.6  438.84
  5083.1  439.04  5193.3  438.46  5223.4  438.60  5236.0  439.29  5328.4  440.45
  5363.7  442.86  5422.2  445.32  5443.8  446.38  5472.2  448.59  5530.9  453.15
#Mann=9,-1,0
  4291.9    0.05       0  4799.4    0.16       0  4896.0    0.07       0
  4902.0    0.16       0  4924.9    0.05       0  4937.6    0.08       0
  5328.4    0.16       0  5422.2    0.05       0  5472.2    0.08       0
Bank Sta=4896,4902
Exp/Cntr=0.3,0.1

Type RM Length L Ch R = 1,18515,349,349,349
BEGIN DESCRIPTION:
WHITE ROCK CREEK 29.2
END DESCRIPTION:
XS GIS Cut Line= 4
      3549768.11     10579162.69      3549195.22     10578960.88
      3548850.17     10579036.83      3548587.08     10579226.61
#Sta/Elev= 30
  4172.3  452.02  4274.1  449.79  4311.0  447.77  4398.6  444.65  4429.5  442.69
  4560.3  438.01  4579.0  437.65  4602.8  438.25  4634.6  437.79  4646.2  437.06
  4674.6  437.14  4739.2  437.07  4772.8  437.21  4794.9  437.18  4834.1  436.96
  4851.2  437.77  4885.3  436.98  4936.5  437.69  4957.0  437.13  5139.9  436.86
  5142.7  436.36  5145.9  436.86  5166.2  437.32  5220.1  440.98  5285.6  446.34
  5321.2  447.12  5335.9  448.07  5356.8  447.91  5392.4  448.89  5457.4  451.72
#Mann=9,-1,0
  4172.3    0.05       0  4674.6    0.16       0  4739.2    0.05       0
  4772.8    0.16       0  4794.9    0.08       0  5139.9    0.07       0
  5145.9    0.08       0  5166.2    0.16       0  5220.1    0.05       0
Bank Sta=5139.9,5145.9
Exp/Cntr=0.3,0.1

Type RM Length L Ch R = 1,18166,596,596,596
BEGIN DESCRIPTION:
WHITE ROCK CREEK 29.0
END DESCRIPTION:
XS GIS Cut Line= 5
      3549896.43     10579183.89      3548950.29     10578645.72
      3548737.62     10578728.19      3548542.11     10579191.64
      3548436.28     10579265.76
#Sta/Elev= 30
  3819.8  453.89  3934.8  452.15  4080.4  445.52  4204.4  440.98  4419.1  437.86
  4534.8  437.31  4592.2  436.94  4728.1  437.19  4756.6  437.07  4806.9  438.37
  4839.4  436.94  4930.7  436.96  4981.4  436.95  5013.6  437.91  5035.1  436.31
  5096.3  435.75  5099.0  435.25  5102.3  435.75  5224.8  436.37  5289.4  436.50
  5418.8  443.97  5500.8  445.12  5630.3  451.13  5646.8  450.78  5667.7  451.66
  5682.6  450.85  5703.5  451.47  5733.1  450.23  5739.2  450.69  5768.6  450.04
#Mann=9,-1,0
  3819.8    0.05       0  4534.8    0.16       0  4592.2    0.05       0
  4728.1    0.08       0  4839.4    0.05       0  4930.7    0.08       0
  5096.3    0.07       0  5102.3    0.08       0  5224.8    0.05       0
Bank Sta=5096.3,5102.3
Exp/Cntr=0.3,0.1

Type RM Length L Ch R = 1,17570,454,454,454
BEGIN DESCRIPTION:
WHITE ROCK CREEK 29.1
END DESCRIPTION:
XS GIS Cut Line= 3
      3549650.65     10577864.48      3548374.64     10578220.37
      3547525.55     10578259.36
#Sta/Elev= 30
  4088.2  451.65  4117.5  450.76  4149.0  448.35  4190.5  448.06  4467.1  437.28
  4969.1  435.30  4979.5  434.71  4987.1  430.23  4992.3  431.62  4997.3  428.43
  5000.0  427.93  5003.3  428.43  5010.7  428.84  5021.0  434.48  5026.5  435.61
  5260.3  434.17  5280.6  434.64  5286.6  429.53  5291.8  429.31  5311.7  434.38
  5374.0  434.36  5399.5  432.01  5455.5  438.15  5475.5  438.38  5585.6  446.44
  5663.3  455.04  5725.8  457.39  5946.0  459.53  5983.3  461.24  6262.9  462.55
#Mann=6,-1,0
  4088.2    0.08       0  4117.5    0.05       0  4997.3    0.04       0
  5003.3    0.05       0  5260.3    0.16       0  5663.3    0.05       0
Bank Sta=4997.3,5003.3
Exp/Cntr=0.3,0.1

Type RM Length L Ch R = 1,17116,11,11,11
BEGIN DESCRIPTION:
WHITE ROCK CREEK 28.03
END DESCRIPTION:
XS GIS Cut Line= 6
      3549618.41     10577848.74      3549479.53     10577886.93
      3549252.10     10577836.58      3548503.84     10577850.47
      3548279.88     10577897.34      3547578.54     10577945.95
#Sta/Elev= 30
  3853.8  450.66  3908.0  448.99  3932.9  446.47  3997.3  445.16  4077.1  440.57
  4228.1  437.44  4690.8  434.16  4910.9  434.66  4920.9  434.47  4940.9  431.82
  4950.9  433.34  4970.9  432.90  4982.6  432.07  4998.4  429.13  5001.1  428.63
  5004.4  429.13  5021.8  432.98  5042.2  433.15  5052.5  433.93  5057.8  435.56
  5062.9  434.68  5083.1  438.22  5102.7  439.64  5107.8  439.11  5137.1  440.52
  5225.8  444.65  5265.9  448.56  5436.3  453.86  5596.7  454.37  5911.0  458.13
#Mann=5,-1,0
  3853.8    0.08       0  3908.0    0.05       0  4998.4    0.04       0
  5004.4    0.05       0  5137.1    0.08       0
Bank Sta=4998.4,5004.4
Exp/Cntr=0.3,0.1

Type RM Length L Ch R = 1,17105,80,80,80
BEGIN DESCRIPTION:
WHITE ROCK CREEK 28.02
END DESCRIPTION:
XS GIS Cut Line= 6
      3549594.09     10577841.80      3549470.85     10577869.57
      3549245.16     10577815.75      3548486.48     10577843.52
      3548283.35     10577879.98      3547556.50     10577930.29
#Sta/Elev= 30
  3874.8  449.84  3942.9  446.87  3969.1  444.84  4001.1  444.72  4056.6  441.12
  4098.7  439.72  4254.4  436.92  4359.1  436.39  4526.2  434.36  4609.4  434.52
  4802.9  433.21  4807.9  434.60  4836.6  434.75  4926.7  432.70  4976.7  433.77
  4986.7  432.16  4992.0  429.18  5002.9  428.48  5005.7  427.98  5008.9  428.48
  5017.1  431.49  5037.4  431.85  5069.8  437.73  5131.2  440.85  5290.2  447.42
  5310.2  449.46  5437.7  452.63  5450.6  453.72  5727.9  455.29  5927.3  457.94
#Mann=7,-1,0
  3874.8    0.08       0  3942.9    0.05       0  4359.1    0.08       0
  4609.4    0.05       0  5002.9    0.04       0  5008.9    0.05       0
  5131.2    0.08       0
Bank Sta=5002.9,5008.9
Exp/Cntr=0.3,0.1

Type RM Length L Ch R = 1,17025,59,59,59
BEGIN DESCRIPTION:
WHITE ROCK CREEK 28.0
END DESCRIPTION:
XS GIS Cut Line= 5
      3549830.26     10577867.84      3549215.65     10577725.47
      3548479.53     10577768.87      3548356.27     10577794.91
      3547538.59     10577836.58
#Sta/Elev= 30
  3586.2  454.86  3645.9  455.92  3675.8  454.53  3681.0  455.33  3723.7  452.40
  3728.8  452.99  3814.2  450.56  3912.8  444.99  3990.0  444.23  4015.4  442.53
  4075.4  440.97  4087.3  439.71  4216.3  436.55  4683.5  433.11  4962.1  433.96
  4972.3  433.61  4982.5  431.55  4992.0  427.25  4994.7  426.75  4998.0  427.25
  5023.4  431.35  5033.6  431.76  5044.7  434.89  5084.0  437.52  5274.9  445.03
  5415.1  451.84  5503.8  451.95  5545.2  453.24  5635.3  451.96  5899.2  454.95
#Mann=5,-1,0
  3586.2    0.08       0  4683.5    0.05       0  4992.0    0.04       0
  4998.0    0.05       0  5084.0    0.08       0
Bank Sta=4992,4998
Exp/Cntr=0.3,0.1

Type RM Length L Ch R = 1,16966,721,721,721
BEGIN DESCRIPTION:
WHITE ROCK CREEK 28.01
END DESCRIPTION:
XS GIS Cut Line= 3
      3549809.43     10577822.70      3549239.95     10577687.27
      3547529.88     10577767.14
#Sta/Elev= 30
  3586.9  456.24  3653.6  456.96  3738.0  450.40  3743.1  449.29  3785.3  447.58
  3790.4  446.47  3933.6  443.16  3954.0  444.03  3974.8  442.17  3995.3  442.08
  4109.1  437.70  4313.9  434.73  4661.0  432.52  4880.9  432.98  4930.9  434.44
  4971.0  433.27  4981.0  431.94  4998.0  427.49  5000.8  426.99  5004.0  427.49
  5011.0  428.37  5016.1  432.28  5021.1  431.65  5031.0  434.30  5131.2  437.02
  5331.4  445.76  5491.5  451.39  5601.7  450.13  5681.8  451.52  5884.2  452.89
#Mann=6,-1,0
  3586.9    0.08       0  4109.1    0.05       0  4313.9    0.08       0
  4661.0    0.05       0  4998.0    0.03       0  5004.0    0.05       0
Bank Sta=4998,5004
Exp/Cntr=0.3,0.1

Type RM Length L Ch R = 1,16245,1110,1110,1110
BEGIN DESCRIPTION:
WHITE ROCK CREEK 26.0
END DESCRIPTION:
XS GIS Cut Line= 4
      3549649.06     10576393.13      3548537.97     10576948.67
      3548255.85     10577087.56      3546750.79     10577516.96
#Sta/Elev= 30
  3591.1  476.70  3744.2  474.20  3842.1  469.88  4266.9  443.58  4451.4  434.40
  4557.6  431.99  4705.7  430.64  4786.8  431.43  4833.3  430.70  4966.3  432.29
  4988.8  431.32  5002.7  427.48  5005.4  426.98  5008.7  427.48  5018.2  431.57
  5045.2  431.89  5101.1  430.25  5145.2  431.48  5179.3  430.42  5291.1  432.63
  5463.7  433.08  5588.4  436.47  5801.1  439.24  5980.6  446.55  6019.6  446.88
  6170.8  453.53  6199.1  453.41  6337.2  456.81  6649.1  466.94  6712.9  467.75
#Mann=5,-1,0
  3591.1    0.05       0  5002.7    0.03       0  5008.7    0.05       0
  5045.2    0.16       0  5145.2    0.05       0
Bank Sta=5002.7,5008.7
Exp/Cntr=0.3,0.1

Type RM Length L Ch R = 1,15135,719,719,719
BEGIN DESCRIPTION:
WHITE ROCK CREEK 24.0
END DESCRIPTION:
XS GIS Cut Line= 3
      3548592.10     10575991.65      3547692.11     10576391.64
      3546492.12     10576991.64
#Sta/Elev= 30
  4037.5  452.98  4114.1  451.55  4347.3  441.94  4431.4  436.69  4544.3  433.32
  4567.6  433.27  4637.3  430.64  4741.3  428.76  4908.2  429.51  4984.8  430.16
  5000.5  425.64  5005.0  425.03  5007.8  424.53  5011.0  425.03  5019.6  429.70
  5067.1  428.30  5146.2  428.02  5164.9  428.88  5192.9  428.64  5254.4  429.72
  5401.6  434.55  5478.0  438.24  5577.7  440.52  5656.9  443.57  5930.8  451.61
  6073.3  456.80  6162.8  459.05  6207.5  462.14  6310.9  465.23  6364.0  467.87
#Mann=7,-1,0
  4037.5    0.05       0  4908.2    0.16       0  5005.0    0.07       0
  5011.0    0.16       0  5146.2    0.05       0  5401.6    0.16       0
  5577.7    0.05       0
Bank Sta=5005,5011
Exp/Cntr=0.3,0.1

Type RM Length L Ch R = 1,14416,649,649,649
BEGIN DESCRIPTION:
WHITE ROCK CREEK 23.0
END DESCRIPTION:
XS GIS Cut Line= 3
      3548500.59     10575779.40      3547750.64     10575748.15
      3546629.15     10575584.96
#Sta/Elev= 30
  4119.6  451.65  4158.1  450.20  4228.2  445.59  4348.3  439.84  4588.5  430.21
  4808.7  426.53  4929.9  428.45  4990.0  428.34  4997.1  423.99  4999.8  423.49
  5003.1  423.99  5010.2  426.72  5017.4  428.20  5092.6  426.96  5137.5  427.08
  5252.7  427.42  5358.8  429.27  5503.0  434.77  5508.1  434.22  5573.1  437.23
  5677.1  438.01  5687.3  438.67  5707.5  441.58  5713.3  440.11  5718.3  440.65
  5758.0  439.73  5768.1  441.17  5853.5  446.11  5929.8  452.51  6003.5  456.53
#Mann=5,-1,0
  4119.6    0.05       0  4929.9    0.16       0  4997.1    0.07       0
  5003.1    0.16       0  5137.5    0.05       0
Bank Sta=4997.1,5003.1
Exp/Cntr=0.3,0.1

Type RM Length L Ch R = 1,13767,930,930,930
BEGIN DESCRIPTION:
WHITE ROCK CREEK 21.0
END DESCRIPTION:
XS GIS Cut Line= 3
      3548342.08     10575291.64      3547742.11     10575141.64
      3547192.09     10574941.64
#Sta/Elev= 30
  4382.6  444.62  4441.8  442.87  4578.4  441.00  4611.9  439.33  4689.2  432.51
  4812.9  426.37  4859.3  426.05  4941.8  427.32  4977.9  426.59  4984.6  425.34
  4995.5  422.67  4998.2  422.17  5001.5  422.67  5003.7  422.67  5016.3  427.54
  5088.9  426.55  5213.9  425.49  5281.0  425.78  5288.3  426.63  5311.6  425.16
  5330.9  425.84  5336.9  426.92  5367.5  428.27  5398.1  430.88  5423.3  434.86
  5448.0  437.55  5453.9  438.75  5522.4  447.66  5540.4  449.51  5586.3  452.44
#Mann=5,-1,0
  4382.6    0.05       0  4984.6    0.16       0  4995.5    0.07       0
  5001.5    0.16       0  5088.9    0.05       0
Bank Sta=4995.5,5001.5
Exp/Cntr=0.3,0.1

Type RM Length L Ch R = 1,12837,400,400,400
BEGIN DESCRIPTION:
WHITE ROCK CREEK 20.0
END DESCRIPTION:
XS GIS Cut Line= 2
      3549171.82     10574731.55      3546977.38     10574037.11
#Sta/Elev= 30
  3582.7  449.48  3695.5  445.57  3727.8  445.63  3733.0  448.16  3760.1  444.49
  3765.3  445.75  3771.2  444.18  3797.6  442.08  3835.2  441.70  3862.2  439.74
  3899.8  439.86  3991.5  435.08  4085.9  431.99  4362.6  428.34  4400.5  426.52
  4421.5  427.32  4820.1  424.56  4966.9  426.35  4977.4  425.88  4995.4  421.66
  4998.1  421.16  5001.4  421.66  5019.2  425.39  5089.3  425.39  5176.7  424.87
  5239.6  427.59  5616.4  432.24  5711.6  437.22  5827.0  448.56  5884.4  450.08
#Mann=5,-1,0
  3582.7    0.05       0  4820.1    0.16       0  4995.4    0.07       0
  5001.4    0.16       0  5089.3    0.05       0
Bank Sta=4995.4,5001.4
Exp/Cntr=0.3,0.1

Type RM Length L Ch R = 1,12437,757,757,757
BEGIN DESCRIPTION:
WHITE ROCK CREEK 18.0
END DESCRIPTION:
XS GIS Cut Line= 3
      3549092.08     10574341.63      3547892.11     10573941.64
      3547342.13     10573691.66
#Sta/Elev= 30
  3714.0  459.55  3724.5  459.81  3735.1  457.22  3756.1  455.11  3766.7  451.59
  3798.3  447.24  3808.8  446.42  3924.8  438.98  4114.5  429.63  4262.1  426.54
  4430.8  424.51  4567.8  423.71  4873.5  423.51  4958.8  425.20  4987.7  424.67
  4997.8  420.75  5000.6  420.25  5003.8  420.75  5010.7  423.60  5016.2  424.82
  5022.8  425.31  5086.5  424.30  5108.5  423.77  5114.0  424.42  5234.8  425.20
  5350.2  428.80  5418.3  434.47  5528.1  447.73  5568.8  451.64  5583.0  452.11
#Mann=5,-1,0
  3714.0    0.05       0  4958.8    0.16       0  4997.8    0.07       0
  5003.8    0.16       0  5086.5    0.05       0
Bank Sta=4997.8,5003.8
Exp/Cntr=0.3,0.1

Type RM Length L Ch R = 1,11680,502,502,502
BEGIN DESCRIPTION:
WHITE ROCK CREEK 17.0
END DESCRIPTION:
XS GIS Cut Line= 4
      3549615.21     10573140.51      3548292.31     10573338.43
      3547945.08     10573477.32      3547592.07     10573491.64
#Sta/Elev= 30
  3586.9  470.01  3620.4  469.21  3626.9  467.80  3631.9  468.87  3782.2  466.86
  3898.5  460.23  3974.3  457.91  4031.9  458.24  4055.2  457.25  4176.5  445.07
  4303.5  435.46  4388.8  433.53  4540.5  427.67  4682.1  423.90  4864.1  421.40
  4978.8  424.36  4990.6  422.31  5000.0  419.59  5002.8  419.09  5006.0  419.59
  5010.9  422.43  5021.7  424.33  5098.8  423.87  5140.3  422.79  5184.1  424.17
  5207.0  424.88  5242.6  426.55  5341.5  428.50  5481.6  433.66  5651.8  444.07
#Mann=7,-1,0
  3586.9    0.05       0  4990.6    0.16       0  5000.0    0.07       0
  5006.0    0.16       0  5098.8    0.05       0  5184.1    0.16       0
  5207.0    0.05       0
Bank Sta=5000,5006
Exp/Cntr=0.3,0.1

Type RM Length L Ch R = 1,11178,44,44,44
BEGIN DESCRIPTION:
WHITE ROCK CREEK 15.03
END DESCRIPTION:
XS GIS Cut Line= 6
      3548681.97     10572655.12      3548351.06     10572700.69
      3548174.20     10572893.83      3548119.94     10572893.83
      3547893.16     10573150.99      3547406.57     10573418.67
#Sta/Elev= 30
  4375.9  465.54  4455.9  463.14  4517.1  455.61  4538.0  451.51  4547.4  451.25
  4638.2  439.50  4823.0  423.62  4887.1  421.74  4929.0  422.29  4950.6  420.44
  4957.4  420.66  4964.8  422.82  4983.9  423.41  4993.9  420.15  5000.9  419.30
  5003.7  418.80  5006.9  419.30  5022.5  423.76  5028.8  423.56  5058.5  424.41
  5102.5  423.53  5185.7  422.85  5277.7  430.55  5323.1  431.70  5342.2  432.63
  5348.8  434.48  5378.3  435.78  5650.1  436.14  5718.1  438.28  5924.3  441.21
#Mann=7,-1,0
  4375.9    0.05       0  5000.9    0.03       0  5006.9    0.05       0
  5028.8    0.16       0  5102.5    0.05       0  5323.1     0.1       0
  5718.1    0.05       0
Bank Sta=5000.9,5006.9
Exp/Cntr=0.3,0.1

Type RM Length L Ch R = 1,11134,74,74,74
BEGIN DESCRIPTION:
WHITE ROCK CREEK 15.02
END DESCRIPTION:
XS GIS Cut Line= 6
      3548652.67     10572639.93      3548340.21     10572673.56
      3548170.94     10572847.17      3548098.24     10572888.41
      3547897.50     10573100.00      3547382.68     10573396.97
#Sta/Elev= 30
  4424.8  465.65  4489.1  462.93  4576.1  452.85  4616.5  445.91  4646.6  443.37
  4696.9  436.21  4786.1  428.38  4884.8  422.60  4906.4  423.89  4914.4  423.02
  4920.4  424.55  4935.4  422.70  4941.4  424.04  4950.3  423.11  4956.4  424.77
  5004.8  419.23  5007.5  418.73  5010.8  419.23  5017.6  419.45  5023.9  421.89
  5029.9  421.11  5047.1  423.08  5092.2  423.51  5208.2  422.85  5292.6  429.17
  5328.3  431.04  5377.1  435.85  5655.7  435.83  5722.0  437.05  5953.0  440.57
#Mann=7,-1,0
  4424.8    0.05       0  5004.8    0.03       0  5010.8    0.05       0
  5047.1    0.16       0  5092.2    0.05       0  5292.6     0.1       0
  5722.0    0.05       0
Bank Sta=5004.8,5010.8
Exp/Cntr=0.3,0.1

Type RM Length L Ch R = 1,11060,41,41,41
BEGIN DESCRIPTION:
WHITE ROCK CREEK 15.0
END DESCRIPTION:
XS GIS Cut Line= 6
      3548612.37     10572537.93      3548323.76     10572624.73
      3548165.52     10572775.56      3548125.37     10572786.41
      3547859.53     10573078.29      3547348.45     10573371.27
#Sta/Elev= 30
  4462.6  460.05  4506.0  456.59  4573.8  453.14  4762.2  431.47  4911.5  422.65
  4975.0  423.99  4984.7  422.18  4989.0  423.89  4996.5  419.53  5003.8  418.52
  5006.6  418.02  5009.8  418.52  5023.3  423.24  5051.6  424.16  5115.3  423.11
  5129.6  424.20  5164.8  422.73  5221.5  423.22  5228.8  424.47  5235.6  422.89
  5249.8  423.04  5257.1  424.38  5264.0  422.81  5361.7  429.91  5434.7  433.20
  5440.4  435.19  5462.2  436.44  5743.8  436.55  5831.1  436.78  6008.2  440.42
#Mann=7,-1,0
  4462.6    0.05       0  4506.0    0.16       0  4573.8    0.05       0
  5003.8    0.03       0  5009.8    0.05       0  5361.7     0.1       0
  5743.8    0.05       0
Bank Sta=5003.8,5009.8
Exp/Cntr=0.3,0.1

Type RM Length L Ch R = 1,11019,747,747,747
BEGIN DESCRIPTION:
WHITE ROCK CREEK 15.01
END DESCRIPTION:
XS GIS Cut Line= 5
      3548612.55     10572514.06      3548307.66     10572595.44
      3548121.03     10572758.20      3547794.42     10573081.55
      3547337.61     10573344.14
#Sta/Elev= 30
  4461.0  459.33  4487.3  457.10  4508.9  454.29  4514.1  455.26  4543.8  452.09
  4589.1  450.55  4664.1  442.24  4704.2  439.29  4739.1  434.13  4792.1  429.10
  4912.7  422.52  4976.2  422.18  4983.0  419.49  4994.1  417.75  4996.9  417.25
  5000.1  417.75  5013.7  420.61  5019.0  423.35  5054.1  423.85  5167.3  422.50
  5301.7  423.07  5416.5  429.49  5457.2  431.07  5478.4  435.31  5498.9  436.43
  5552.1  436.90  5632.6  435.17  5737.9  436.24  5821.0  436.21  6010.7  440.09
#Mann=9,-1,0
  4461.0    0.05       0  4487.3    0.16       0  4664.1    0.05       0
  4976.2    0.16       0  4994.1    0.07       0  5000.1    0.16       0
  5013.7    0.05       0  5416.5     0.1       0  5737.9    0.05       0
Bank Sta=4994.1,5000.1
Exp/Cntr=0.3,0.1

Type RM Length L Ch R = 1,10272,699,699,699
BEGIN DESCRIPTION:
WHITE ROCK CREEK 14.0
END DESCRIPTION:
XS GIS Cut Line= 4
      3549184.71     10572109.26      3548000.64     10572244.68
      3547577.03     10572421.76      3547090.96     10572609.25
#Sta/Elev= 30
  3714.8  468.07  3767.7  465.29  3781.3  466.87  3838.2  465.04  4005.1  456.74
  4160.3  449.10  4200.6  449.37  4250.9  446.79  4307.0  439.86  4361.6  439.45
  4391.3  434.40  4396.3  435.30  4422.0  433.24  4442.1  433.97  4480.6  432.43
  4485.6  435.34  4553.3  432.72  4794.4  421.81  4931.1  421.42  4980.9  422.23
  4999.5  417.01  5002.3  416.51  5005.5  417.01  5011.7  419.76  5024.2  422.09
  5157.5  422.28  5223.8  422.05  5348.2  432.44  5716.0  439.57  5886.7  444.76
#Mann=7,-1,0
  3714.8    0.05       0  4005.1    0.16       0  4553.3    0.05       0
  4931.1    0.16       0  4999.5    0.07       0  5005.5    0.16       0
  5157.5    0.05       0
Bank Sta=4999.5,5005.5
Exp/Cntr=0.3,0.1

Type RM Length L Ch R = 1,9573,1057,1057,1057
BEGIN DESCRIPTION:
WHITE ROCK CREEK 12.0
END DESCRIPTION:
XS GIS Cut Line= 3
      3548735.14     10571425.68      3547735.16     10571725.67
      3547136.13     10571825.51
#Sta/Elev= 30
  3959.0  463.66  3964.9  464.53  3992.7  461.04  3997.9  461.56  4031.0  456.86
  4036.2  457.05  4064.1  453.85  4102.3  451.22  4135.4  446.35  4168.5  443.17
  4206.7  440.96  4239.8  437.76  4448.6  422.04  4514.7  420.47  4630.3  419.58
  4975.8  420.76  4985.3  420.61  4997.5  418.32  5002.0  416.48  5007.1  416.25
  5009.8  415.75  5013.1  416.25  5026.4  420.12  5036.5  421.27  5178.5  419.72
  5253.7  419.96  5360.9  420.20  5462.3  430.03  5563.7  436.02  5610.3  437.43
#Mann=5,-1,0
  3959.0    0.05       0  4997.5    0.16       0  5007.1    0.07       0
  5013.1    0.16       0  5253.7    0.05       0
Bank Sta=5007.1,5013.1
Exp/Cntr=0.3,0.1

Type RM Length L Ch R = 1,8516,778,778,778
BEGIN DESCRIPTION:
WHITE ROCK CREEK 10.0
END DESCRIPTION:
XS GIS Cut Line= 3
      3547702.25     10570865.66      3546632.78     10571233.73
      3546529.05     10571537.99
#Sta/Elev= 30
  4351.1  439.52  4435.9  440.10  4449.0  439.43  4467.6  435.03  4475.0  432.51
  4480.2  432.90  4488.7  430.10  4506.2  426.10  4615.6  419.31  4710.8  417.62
  4906.0  418.84  4975.2  419.99  4985.8  418.44  4992.3  415.15  4995.0  414.65
  4998.3  415.15  5000.5  415.39  5006.9  418.26  5017.5  420.09  5112.7  417.99
  5169.8  418.61  5219.1  418.84  5375.1  422.60  5387.7  425.32  5395.9  426.13
  5408.8  426.31  5427.2  424.85  5481.2  427.04  5680.5  434.99  5803.6  437.97
#Mann=7,-1,0
  4351.1    0.05       0  4906.0    0.16       0  4992.3    0.07       0
  4998.3    0.16       0  5169.8    0.05       0  5375.1    0.08       0
  5481.2    0.05       0
Bank Sta=4992.3,4998.3
Exp/Cntr=0.3,0.1

Type RM Length L Ch R = 1,7738,33,33,33
BEGIN DESCRIPTION:
WHITE ROCK CREEK 9.0
END DESCRIPTION:
XS GIS Cut Line= 4
      3548271.72     10570540.93      3547245.28     10570471.49
      3547158.47     10570501.87      3546295.92     10570439.02
#Sta/Elev= 30
  3945.0  443.85  4115.0  439.85  4307.6  434.17  4395.6  434.18  4435.7  433.32
  4451.9  434.05  4456.9  433.16  4495.9  432.81  4525.9  430.97  4606.1  428.10
  4750.4  425.07  4846.7  419.00  4894.6  417.75  4906.8  418.53  4985.9  418.14
  4995.3  414.54  4998.1  414.04  5001.3  414.54  5008.9  415.25  5017.0  418.04
  5022.2  418.33  5102.2  417.23  5372.9  417.01  5393.0  419.47  5462.7  419.02
  5513.3  420.24  5633.6  425.49  5723.9  428.35  5804.1  430.18  5930.6  431.66
#Mann=4,-1,0
  3945.0    0.08       0  4995.3    0.07       0  5001.3    0.08       0
  5462.7    0.05       0
Bank Sta=4995.3,5001.3
Exp/Cntr=0.3,0.1

Type RM Length L Ch R = 1,7705,75,75,75
BEGIN DESCRIPTION:
WHITE ROCK CREEK 8.0
END DESCRIPTION:
XS GIS Cut Line= 4
      3548275.29     10570511.85      3547226.92     10570445.44
      3547157.48     10570468.23      3546266.79     10570402.06
#Sta/Elev= 30
  3920.5  442.62  4104.1  438.61  4204.3  434.69  4354.6  432.81  4394.6  430.56
  4444.7  431.11  4454.8  429.55  4473.6  431.41  4555.0  428.01  4725.3  425.72
  4792.1  421.19  4827.1  420.58  4939.7  419.16  4956.4  419.54  4978.1  418.19
  4994.1  413.83  4996.8  413.33  5000.1  413.83  5011.7  416.82  5028.7  418.06
  5320.2  416.78  5330.2  416.91  5340.4  418.96  5369.5  419.24  5420.5  418.80
  5500.7  420.21  5711.3  427.70  5801.5  428.68  5841.6  430.45  5937.2  430.93
#Mann=7,-1,0
  3920.5    0.08       0  4827.1    0.05       0  4939.7    0.16       0
  4994.1    0.07       0  5000.1    0.16       0  5011.7    0.08       0
  5369.5    0.05       0
Bank Sta=4994.1,5000.1
Exp/Cntr=0.3,0.1

Type RM Length L Ch R = 1,7630,27,27,27
BEGIN DESCRIPTION:
WHITE ROCK CREEK 7.0
END DESCRIPTION:
XS GIS Cut Line= 3
      3548251.85     10570444.14      3547100.84     10570392.06
      3546228.41     10570353.00
#Sta/Elev= 30
  3906.8  439.66  4136.8  434.20  4256.9  429.96  4297.9  430.50  4467.1  426.94
  4697.4  425.01  4777.4  421.26  4899.6  420.04  4955.1  419.92  4960.1  418.72
  4977.6  418.55  4987.7  415.50  4994.7  410.86  4997.4  410.36  5000.7  410.86
  5027.7  417.35  5047.7  418.54  5107.8  418.15  5117.8  415.91  5137.8  414.90
  5157.8  416.25  5196.1  415.71  5318.0  417.05  5403.4  420.60  5408.4  419.41
  5438.1  419.76  5568.2  424.16  5847.1  430.31  5878.5  429.84  5932.3  430.89
#Mann=5,-1,0
  3906.8    0.05       0  4899.6    0.16       0  4994.7    0.07       0
  5000.7    0.16       0  5196.1    0.05       0
Bank Sta=4994.7,5000.7
Exp/Cntr=0.3,0.1

Type RM Length L Ch R = 1,7603,820,820,820
BEGIN DESCRIPTION:
WHITE ROCK CREEK 6.0
END DESCRIPTION:
XS GIS Cut Line= 4
      3548267.45     10570420.70      3547246.67     10570371.23
      3547020.11     10570366.02      3546255.81     10570327.02
#Sta/Elev= 30
  3881.7  439.52  4037.2  435.23  4097.3  435.05  4227.5  431.34  4247.5  429.31
  4287.5  430.58  4597.9  424.00  4698.0  425.74  4798.1  419.75  4889.2  418.55
  4968.3  417.21  4978.3  415.00  4988.3  410.65  4995.3  410.36  4998.0  409.86
  5001.3  410.36  5028.3  414.60  5058.3  417.18  5088.3  417.41  5098.2  411.26
  5103.2  411.06  5108.3  416.24  5118.3  417.44  5185.7  417.96  5278.5  417.03
  5418.7  419.97  5448.7  419.32  5578.9  423.93  5710.4  425.49  5895.6  430.23
#Mann=5,-1,0
  3881.7    0.05       0  4889.2    0.16       0  4995.3    0.07       0
  5001.3    0.16       0  5185.7    0.05       0
Bank Sta=4995.3,5001.3
Exp/Cntr=0.3,0.1

Type RM Length L Ch R = 1,6783,719,719,719
BEGIN DESCRIPTION:
WHITE ROCK CREEK 6.1
END DESCRIPTION:
XS GIS Cut Line= 3
      3548161.54     10570215.17      3547557.34     10569916.54
      3546246.01     10569826.34
#Sta/Elev= 30
  3659.0  430.56  3727.1  429.03  3974.0  426.30  4086.2  426.89  4243.2  426.04
  4310.5  423.60  4368.3  419.88  4418.4  417.54  4438.5  417.50  4458.5  415.88
  4749.2  415.88  4789.3  415.14  4808.8  415.68  4979.7  415.83  4996.8  409.08
  4999.5  408.58  5002.8  409.08  5009.8  412.14  5019.8  415.05  5039.9  417.30
  5049.9  417.06  5069.9  414.10  5085.7  415.15  5110.0  415.59  5140.1  417.74
  5205.5  419.68  5430.8  420.54  5500.9  422.76  5581.1  424.80  5647.4  424.99
#Mann=6,-1,0
  3659.0    0.05       0  4808.8    0.16       0  4996.8    0.07       0
  5002.8    0.16       0  5085.7    0.05       0  5500.9    0.16       0
Bank Sta=4996.8,5002.8
Exp/Cntr=0.3,0.1

Type RM Length L Ch R = 1,6064,685,685,685
BEGIN DESCRIPTION:
WHITE ROCK CREEK 5.0
END DESCRIPTION:
XS GIS Cut Line= 3
      3548403.58     10570178.15      3547125.84     10569205.95
      3545910.51     10569351.79
#Sta/Elev= 30
  3033.2  435.70  3096.7  434.30  3138.3  431.84  3252.7  428.77  3516.7  425.53
  3688.5  422.09  3809.9  421.22  3952.3  418.21  4059.4  417.33  4655.4  416.56
  4692.9  414.98  4773.4  413.79  4974.9  414.70  4980.1  413.50  4985.1  413.66
  4995.0  410.78  5002.1  407.43  5004.8  406.93  5008.1  407.43  5015.2  408.21
  5035.3  414.75  5055.8  416.07  5319.2  419.36  5456.1  423.57  5559.0  426.61
  5589.3  429.05  5619.5  429.36  5659.8  432.21  5740.5  435.70  5862.8  437.04
#Mann=6,-1,0
  3033.2    0.05       0  4655.4    0.16       0  5002.1    0.07       0
  5008.1    0.16       0  5055.8    0.05       0  5456.1    0.16       0
Bank Sta=5002.1,5008.1
Exp/Cntr=0.3,0.1

Type RM Length L Ch R = 1,5379,890,890,890
BEGIN DESCRIPTION:
WHITE ROCK CREEK 3.0
END DESCRIPTION:
XS GIS Cut Line= 4
      3548531.80     10569991.38      3546995.31     10568783.02
      3546870.31     10568616.35      3545797.43     10568809.05
#Sta/Elev= 30
  2728.2  437.72  2962.8  431.44  3041.4  426.61  3275.5  422.32  3817.6  417.00
  3960.4  418.38  4273.1  417.67  4521.6  414.97  4579.4  413.86  4714.6  414.17
  4750.0  413.70  4772.1  412.19  4793.7  413.80  4885.4  412.75  4980.9  413.12
  4991.0  412.40  4998.1  407.84  5000.8  407.34  5004.1  407.84  5011.3  407.97
  5031.7  413.32  5397.2  412.20  5523.8  412.85  5661.6  411.85  5685.9  413.39
  5702.2  412.83  5798.4  416.29  5910.8  423.57  5969.0  425.39  5981.3  425.61
#Mann=6,-1,0
  2728.2    0.05       0  4521.6    0.16       0  4998.1    0.07       0
  5004.1    0.16       0  5523.8    0.05       0  5969.0    0.16       0
Bank Sta=4998.1,5004.1
Exp/Cntr=0.3,0.1

Type RM Length L Ch R = 1,4489,834,834,834
BEGIN DESCRIPTION:
WHITE ROCK CREEK 2.0
END DESCRIPTION:
XS GIS Cut Line= 4
      3548287.07     10567489.48      3546657.49     10567747.56
      3546261.39     10568026.67      3545766.58     10568662.85
#Sta/Elev= 30
  3139.8  450.88  3188.0  451.39  3250.3  449.31  3375.0  440.05  3567.1  428.62
  3742.2  420.77  4013.6  411.55  4258.5  411.90  4335.4  409.90  4714.1  408.44
  4967.7  410.97  4982.5  406.96  4991.2  408.07  4994.3  404.58  4997.0  404.08
  5000.3  404.58  5004.2  405.10  5012.1  409.74  5033.0  410.84  5126.6  409.03
  5241.1  410.05  5270.7  408.94  5377.3  411.57  5505.8  411.74  5655.1  419.00
  5704.8  422.92  5918.4  428.49  5997.1  428.70  6061.4  430.93  6080.2  432.89
#Mann=3,-1,0
  3139.8    0.05       0  4994.3    0.03       0  5000.3    0.05       0
Bank Sta=4994.3,5000.3
Exp/Cntr=0.3,0.1

Type RM Length L Ch R = 1,3655,0,0,0
BEGIN DESCRIPTION:
WHITE ROCK CREEK 1.0
END DESCRIPTION:
XS GIS Cut Line= 5
      3548185.10     10566847.68      3546397.73     10567099.43
      3545983.76     10567295.22      3545852.30     10567395.91
      3545656.81     10568479.48
#Sta/Elev= 30
  2865.3  453.52  3002.9  450.90  3110.7  446.42  3140.3  443.31  3231.9  438.58
  3262.2  433.49  3287.7  430.80  3430.1  420.50  3501.3  416.83  3767.1  409.60
  4864.6  406.85  4986.0  408.84  4991.5  408.08  4997.3  404.86  5005.4  404.58
  5008.1  404.08  5011.4  404.58  5014.3  407.89  5052.6  409.09  5074.8  407.20
  5105.3  406.95  5133.6  408.34  5421.6  409.30  5489.9  410.06  5548.5  412.41
  5602.1  411.90  5714.3  414.07  6109.6  433.82  6356.4  440.69  6394.9  440.60
#Mann=3,-1,0
  2865.3    0.05       0  5005.4    0.03       0  5011.4    0.05       0
Bank Sta=5005.4,5011.4
Exp/Cntr=0.3,0.1

Chan Stop Cuts=-1
