--- WICKSON CREEK.prj (project) ---

Proj Title=WICKSON CREEK Base Level Engineering
Current Plan=p01
Default Exp/Contr=0.3,0.1
English Units
Geom File=g01
Flow File=f01
Plan File=p01
Y Axis Title=Elevation
X Axis Title(PF)=Main Channel Distance
X Axis Title(XS)=Station
BEGIN DESCRIPTION:
WICKSON CREEK
END DESCRIPTION:
DSS Export Rating Curves= 0
DSS Export Rating Curve Sorted= 0
DSS Export Volume Flow Curves= 0
DXF OffsetX= 0
DXF OffsetY= 0
DXF ScaleX= 1
DXF ScaleY= 10

--- WICKSON CREEK.p01 (plan) ---

Plan Title=Multiple Run
Short Identifier=Multiple
Geom File=g01
Flow File=f01
Subcritical Flow
K Sum by GR= 0
Std Step Tol= 0.01
Critical Tol= 0.01
Num of Std Step Trials= 20
Max Error Tol= 0.3
Flow Tol Ratio= 0.001
Split Flow NTrial= 30
Split Flow Tol= 0.02
Split Flow Ratio= 0.02
Log Output Level= 0
Friction Slope Method= 1
Unsteady Friction Slope Method= 2
Unsteady Bridges Friction Slope Method= 1
Parabolic Critical Depth
Global Vel Dist=  1 , 1 , 1
Global Log Level= 0
CheckData=True
Encroach Param= -1, 0, 0, 0
BEGIN DESCRIPTION:
Multiple Run
END DESCRIPTION:

--- WICKSON CREEK.f01 (steady flow) ---

Flow Title=Multiple
Program Version=4.10
Number of Profiles= 7
Profile Names=10-year,25-year,50-year,1pct_min,100-year,1pct_plu,500-year
River Rch & RM=WICKSON CREEK,Reach-1         ,169685
     519     692     830     730     988    1336    1400
River Rch & RM=WICKSON CREEK,Reach-1         ,167730
    1085    1507    1859    1676    2266    3064    3380
River Rch & RM=WICKSON CREEK,Reach-1         ,166854
    1085    1507    1859    1676    2266    3064    3380
River Rch & RM=WICKSON CREEK,Reach-1         ,162240
    1313    1840    2283    2070    2799    3785    4221
River Rch & RM=WICKSON CREEK,Reach-1         ,160527
    1452    2030    2515    2274    3075    4159    4614
River Rch & RM=WICKSON CREEK,Reach-1         ,145453
    1712    2404    2987    2707    3661    4951    5518
River Rch & RM=WICKSON CREEK,Reach-1         ,139852
    2714    3877    4874    4463    6036    8163    9289
River Rch & RM=WICKSON CREEK,Reach-1         ,132818
    3330    4785    6039    5549    7504   10149   11627
River Rch & RM=WICKSON CREEK,Reach-1         ,130718
    3190    4579    5775    5302    7171    9698   11096
River Rch & RM=WICKSON CREEK,Reach-1         ,125846
    3438    4932    6217    5705    7715   10434   11920
River Rch & RM=WICKSON CREEK,Reach-1         ,117075
    3546    5079    6396    5861    7927   10720   12216
River Rch & RM=WICKSON CREEK,Reach-1         ,114881
    4443    6413    8119    7477   10112   13675   15734
River Rch & RM=WICKSON CREEK,Reach-1         ,111131
    4379    6300    7957    7310    9887   13370   15309
River Rch & RM=WICKSON CREEK,Reach-1         ,107055
    4403    6326    7986    7331    9914   13408   15328
River Rch & RM=WICKSON CREEK,Reach-1         ,99859
    4417    6341    7999    7338    9924   13421   15323
River Rch & RM=WICKSON CREEK,Reach-1         ,91302
    5963    8604   10893   10024   13556   18333   21048
River Rch & RM=WICKSON CREEK,Reach-1         ,86403
    5963    8604   10893   10024   13556   18333   21048
River Rch & RM=WICKSON CREEK,Reach-1         ,83158
    6133    8851   11206   10312   13946   18860   21653
River Rch & RM=WICKSON CREEK,Reach-1         ,73759
    6195    8932   11304   10396   14059   19013   21802
River Rch & RM=WICKSON CREEK,Reach-1         ,70897
    6399    9212   11646   10697   14466   19564   22376
River Rch & RM=WICKSON CREEK,Reach-1         ,68155
    6399    9212   11646   10697   14466   19564   22376
River Rch & RM=WICKSON CREEK,Reach-1         ,57540
    6412    9223   11653   10697   14467   19565   22351
River Rch & RM=WICKSON CREEK,Reach-1         ,53782
    6424    9231   11654   10690   14457   19552   22300
River Rch & RM=WICKSON CREEK,Reach-1         ,51627
    6424    9231   11654   10690   14457   19552   22300
River Rch & RM=WICKSON CREEK,Reach-1         ,49437
    6919    9950   12570   11536   15602   21099   24087
River Rch & RM=WICKSON CREEK,Reach-1         ,42310
    6919    9950   12570   11536   15602   21099   24087
River Rch & RM=WICKSON CREEK,Reach-1         ,26566
    7006   10076   12731   11685   15803   21372   24401
River Rch & RM=WICKSON CREEK,Reach-1         ,25485
    6949    9979   12594   11546   15614   21117   24054
River Rch & RM=WICKSON CREEK,Reach-1         ,22763
    7043   10120   12777   11718   15848   21432   24432
River Rch & RM=WICKSON CREEK,Reach-1         ,19360
    7692   11053   13958   12802   17313   23414   26689
River Rch & RM=WICKSON CREEK,Reach-1         ,16416
    7692   11053   13958   12802   17313   23414   26689
Boundary for River Rch & Prof#=WICKSON CREEK,Reach-1         , 1
Up Type= 0
Dn Type= 3
Dn Slope=0.001
Boundary for River Rch & Prof#=WICKSON CREEK,Reach-1         , 2
Up Type= 0
Dn Type= 3
Dn Slope=0.001
Boundary for River Rch & Prof#=WICKSON CREEK,Reach-1         , 3
Up Type= 0
Dn Type= 3
Dn Slope=0.001
Boundary for River Rch & Prof#=WICKSON CREEK,Reach-1         , 4
Up Type= 0
Dn Type= 3
Dn Slope=0.001
Boundary for River Rch & Prof#=WICKSON CREEK,Reach-1         , 5
Up Type= 0
Dn Type= 3
Dn Slope=0.001
Boundary for River Rch & Prof#=WICKSON CREEK,Reach-1         , 6
Up Type= 0
Dn Type= 3
Dn Slope=0.001
Boundary for River Rch & Prof#=WICKSON CREEK,Reach-1         , 7
Up Type= 0
Dn Type= 3
Dn Slope=0.001
DSS Import GetInterval= 0
DSS Import GetPeak= 0
DSS Import FillOption= 0

--- WICKSON CREEK.g01 (geometry) ---

Geom Title=Existing Conditions
Program Version=4.10

River Reach=WICKSON CREEK   ,Reach-1
Reach XY= 30
      3542762.11     10283081.64      3539932.92     10278194.37
      3542597.44     10271878.89      3545437.19      10269821.1
      3544924.11      10266006.7      3546845.55      10263258.2
      3551981.96     10261071.48      3552943.34     10258274.76
      3568108.42     10252304.46       3569537.6      10248313.7
      3571778.85     10248169.84      3572517.97     10250530.36
       3578434.9     10249596.31      3577792.08     10247631.51
      3580541.27     10247589.38      3580773.01     10245171.56
      3582740.03     10245898.46      3585445.53     10241639.09
      3586559.97     10242342.97      3590498.93     10234705.12
      3592193.42     10236349.29      3593809.02     10235865.05
      3595919.37     10232210.47      3595678.16     10227572.35
       3593800.2      10226807.5      3592634.63     10223653.12
      3598468.66     10219315.59      3597857.62     10218249.01
      3600902.05     10216281.58      3601977.21     10212680.81

Type RM Length L Ch R = 1 ,169685  ,985,985,985
BEGIN DESCRIPTION:
WICKSON CREEK 123.0
END DESCRIPTION:
XS GIS Cut Line= 3
      3543242.12     10282341.63      3542742.11     10282991.64
      3541542.12     10283591.63
#Sta/Elev= 30
  4174.6  365.54    4402  359.68  4609.6  355.36  4624.1   356.2  4638.6  354.93
  4744.6  354.02  4873.2  351.69  4887.8  352.69  4908.6  351.45  4981.1  349.46
  4991.5  347.91  5000.1  347.86  5002.8  347.36  5006.1  347.86  5025.4   349.4
  5053.4   349.9  5084.1  353.61  5218.3  355.11    5249  354.18  5338.5  354.09
  5411.1  354.77  5486.6  356.81  5584.4  358.02  5673.9  356.79  5718.6  356.85
  5813.6  358.92  5875.1  357.73  5956.2  358.15  6269.2  361.59  6336.3  363.14
#Mann= 3 ,-1 , 0
  4174.6     .05       0  5000.1     .03       0  5006.1     .05       0
Bank Sta=4981.1,5025.4
XS Rating Curve= 0 ,0
Exp/Cntr=0.3,0.1

Type RM Length L Ch R = 1 ,168700  ,909,909,909
BEGIN DESCRIPTION:
WICKSON CREEK 121.0
END DESCRIPTION:
XS GIS Cut Line= 3
      3543042.14     10281991.63      3542342.11     10282241.64
      3541442.13     10283441.61
#Sta/Elev= 30
  4234.9  367.15  4306.6  362.87  4406.6  359.19  4486.1  356.09  4573.1  355.03
  4585.4  353.96    4640  353.16  4727.1  353.26  4906.6  349.05  4937.4  347.54
  4981.4  347.08  5011.7  345.92  5014.5  345.42  5017.7  345.92    5021  347.35
  5028.2  347.07    5071   350.4  5085.5  350.33  5091.8  351.15  5114.7  351.35
    5121  352.03    5271  354.12  5414.7  354.75    5521  357.67  5641.8  357.46
    5771  354.77  5956.4  358.73  6050.1  358.64  6356.4  363.87  6478.2  364.91
#Mann= 4 ,-1 , 0
  4234.9      .1       0  4406.6     .05       0  5011.7     .03       0
  5017.7     .05       0
Bank Sta=4981.4,5021
XS Rating Curve= 0 ,0
Exp/Cntr=0.3,0.1

Type RM Length L Ch R = 1 ,167791  ,61,61,61
BEGIN DESCRIPTION:
WICKSON CREEK 119.0
END DESCRIPTION:
XS GIS Cut Line= 3
      3542642.15     10281291.62      3541842.11     10281641.64
       3541442.1     10283041.66
#Sta/Elev= 30
  4143.5  364.03    4148  363.94  4577.4  351.78  4667.5  349.85  4681.9  350.79
  4827.7  347.07  4874.5  347.78  4984.4   345.9  4991.9  344.66  4994.7  344.16
  4997.9  344.66  5002.3   345.7  5072.7  345.83  5172.8  348.71  5224.8  348.03
  5431.5  350.67  5582.3  348.93  5616.1  350.71  5621.3  349.07  5649.9  354.27
  5655.1  352.15  5661.6  354.29    5672  354.81  5688.9  353.03  5694.1  354.65
  5722.7  352.32  5848.8  352.35    5880  354.31    6036  357.62  6472.8  362.23
#Mann= 4 ,-1 , 0
  4143.5      .1       0    4148     .05       0  4991.9     .03       0
  4997.9     .05       0
Bank Sta=4984.4,5002.3
XS Rating Curve= 0 ,0
Exp/Cntr=0.3,0.1

Type RM Length L Ch R = 1 ,167730  ,115,115,115
BEGIN DESCRIPTION:
Mapping XS b863c6ec
END DESCRIPTION:
XS GIS Cut Line= 2
      3542335.74     10281128.14      3541192.52     10282151.58
#Sta/Elev= 30
  4319.6  354.32  4366.9   354.2  4452.1  351.39  4615.1  348.87    4728  348.45
  4784.8  347.17  4905.2  347.36  4926.9  344.62  4947.8  345.65  4982.9  345.83
  4987.4  344.07  4990.2  343.57  4993.4  344.07  5004.6   345.6  5139.2  346.93
  5223.7  346.82  5266.3  347.54  5294.7  348.76  5330.6  347.14  5372.5  347.64
  5521.2  346.34  5599.5  347.34  5613.2   346.6  5620.7  344.86  5634.9  344.45
  5641.6   345.9  5655.8  346.77  5712.6  346.73  5797.9  349.69    5854  350.24
#Mann= 3 ,-1 , 0
  4319.6     .05       0  4987.4     .04       0  4993.4     .05       0
Bank Sta=4982.9,5004.6
XS Rating Curve= 0 ,0
Exp/Cntr=0.3,0.1

Type RM Length L Ch R = 1 ,167615  ,761,761,761
BEGIN DESCRIPTION:
Mapping XS 2ab0189f
END DESCRIPTION:
XS GIS Cut Line= 2
       3542273.2     10281026.62        3541130.     10282073.47
#Sta/Elev= 30
  4321.8  353.19  4496.1  348.72  4693.9  346.57  4714.3  346.39  4843.7  346.02
    4863  346.08  4962.9  346.26  4995.7  342.83  4998.5  342.33  5001.7  342.83
  5027.1  345.77  5076.4  345.31  5113.7  346.18  5139.9  346.71  5393.5  347.76
  5472.9  346.73  5501.3  344.86  5536.4   346.4  5564.8  344.34  5571.6  345.05
    5579  343.74  5585.8   344.9  5593.2  343.59  5599.9  344.53  5614.1  343.61
  5656.7  346.61  5798.5  347.65  5825.8  349.15  5841.1  349.69  5871.9  348.65
#Mann= 11 ,-1 , 0
  4321.8      .1       0  4693.9     .05       0  4714.3     .12       0
  4843.7     .05       0    4863     .12       0  4995.7     .07       0
  5001.7     .12       0  5113.7     .05       0  5139.9     .16       0
  5393.5     .05       0  5825.8      .1       0
Bank Sta=4962.9,5027.1
XS Rating Curve= 0 ,0
Exp/Cntr=0.3,0.1

Type RM Length L Ch R = 1 ,166854  ,948,948,948
BEGIN DESCRIPTION:
WICKSON CREEK 118.0
END DESCRIPTION:
XS GIS Cut Line= 3
      3542042.13     10280191.61      3541442.11     10280991.64
      3540642.13     10281591.62
#Sta/Elev= 30
  4030.8  360.73  4206.2  357.91  4317.3  356.65    4552  346.06    4609   340.3
  4760.1  343.98  4817.3  344.87  4844.4  343.97  4888.1  345.69  4980.8  343.32
  4988.1  340.86  5002.7  341.79    5009  340.41  5017.3  342.54  5020.5  340.28
  5023.3  339.78  5026.5  340.28  5027.7  342.39    5034  342.39  5038.1  340.48
  5044.4  342.39  5052.7  341.99    5059   343.4  5088.1  345.46  5174.9  347.26
  5194.4  348.27  5508.1  348.84  5702.7  352.54    5783   352.6  6030.8  358.28
#Mann= 9 ,-1 , 0
  4030.8     .05       0  4206.2     .16       0    4552     .07       0
  4760.1     .16       0  5020.5     .07       0  5026.5     .16       0
  5174.9     .05       0  5508.1      .1       0    5783     .05       0
Bank Sta=4980.8,5059
XS Rating Curve= 0 ,0
Exp/Cntr=0.3,0.1

Type RM Length L Ch R = 1 ,165906  ,910,910,910
BEGIN DESCRIPTION:
WICKSON CREEK 116.0
END DESCRIPTION:
XS GIS Cut Line= 3
      3541292.09     10280091.65      3541142.11     10280241.64
      3540442.09     10281441.68
#Sta/Elev= 30
  4773.3  353.53  4872.3  346.52  4912.7  345.17    4943  345.05  4957.1  344.04
  4981.9  339.52  4988.3  339.52  4990.3  337.35    4993  336.85  4996.3  337.35
  5014.8  339.44  5020.6  342.23  5036.3     343    5138  341.71  5196.7  343.27
  5233.9  345.63  5263.3  343.38  5341.6  343.65  5511.8  343.95  5576.3  345.77
  5666.4  346.75  5737.9  349.12  5869.8  350.72  5905.7  350.23  6016.9  351.86
  6084.8  352.73  6141.4  353.79  6222.1  356.15  6280.8  356.01  6374.7  358.73
#Mann= 9 ,-1 , 0
  4773.3     .05       0  4912.7     .16       0  4990.3     .07       0
  4996.3     .16       0  5341.6     .05       0  5905.7     .16       0
  6016.9     .05       0  6084.8     .16       0  6141.4     .05       0
Bank Sta=4943,5036.3
XS Rating Curve= 0 ,0
Exp/Cntr=0.3,0.1

Type RM Length L Ch R = 1 ,164996  ,1329,1329,1329
BEGIN DESCRIPTION:
WICKSON CREEK 114.0
END DESCRIPTION:
XS GIS Cut Line= 3
      3541292.06     10279841.66      3540592.11     10280091.64
      3539792.13     10280541.63
#Sta/Elev= 30
    4255   356.9  4506.1  346.99    4588  345.07  4669.1  343.28  4913.8  341.07
  4957.4  340.48  4982.9  338.31  4988.2  339.15  4995.6  336.19  5001.1  336.19
    5009  334.46  5011.7  333.96    5015  334.46  5033.6  338.81  5043.8  339.72
  5049.6  337.52  5065.5  339.93  5108.8  339.84  5181.8  342.53  5280.7  340.96
  5292.4   340.5    5295  339.39  5298.2  338.02    5308  337.82    5330  341.03
  5416.7  343.81  5691.7  345.84  5746.3  347.73  5880.8  349.45  5916.1  350.91
#Mann= 8 ,-1 , 0
    4255     .16       0    4588     .05       0  4913.8     .16       0
    5009     .07       0    5015     .16       0  5280.7     .12       0
    5295     .16       0  5691.7     .05       0
Bank Sta=4988.2,5043.8
XS Rating Curve= 0 ,0
Exp/Cntr=0.3,0.1

Type RM Length L Ch R = 1 ,163667  ,848,848,848
BEGIN DESCRIPTION:
WICKSON CREEK 112.0
END DESCRIPTION:
XS GIS Cut Line= 4
      3541062.37     10279587.22       3540397.8     10279248.53
      3539553.91     10279288.38      3539357.52     10279611.44
#Sta/Elev= 30
  3680.9  351.81  3746.8  350.28    3748  350.25  3846.5  348.94    3879   347.9
  3984.2  347.38  4168.1  344.56  4323.7  344.75  4384.8  343.19  4482.6  342.76
  4582.4  340.15  4628.5  339.67  4692.8  338.77  4782.9  339.94  4822.9  338.93
  4928.1  339.18  4963.1  339.04  4983.1  337.53  5000.1  332.84  5002.9  332.34
  5006.1  332.84  5020.5  337.02  5033.2  338.23  5083.2  336.92  5113.3  337.74
  5117.5  338.48  5133.3  340.79  5173.3  340.65  5319.8  343.77  5649.7  352.19
#Mann= 10 ,-1 , 0
  3680.9      .1       0  3746.8     .16       0    3748      .1       0
  3846.5     .05       0  4582.4     .16       0  4628.5     .05       0
  4928.1     .16       0  5000.1     .07       0  5006.1     .16       0
  5117.5     .05       0
Bank Sta=4963.1,5033.2
XS Rating Curve= 0 ,0
Exp/Cntr=0.3,0.1

Type RM Length L Ch R = 1 ,162819  ,579,579,579
BEGIN DESCRIPTION:
WICKSON CREEK 110.0
END DESCRIPTION:
XS GIS Cut Line= 3
      3541142.08     10279491.62      3539942.11     10278491.64
      3539142.12     10277991.65
#Sta/Elev= 30
  3464.9  351.36  3577.2  349.67  3848.2  345.36  3883.4  343.04  3975.8  343.31
  3990.1  344.62  4181.3  344.07    4296   346.1  4340.7  344.86  4657.9  336.32
  4764.6  337.82  4876.7  337.11  4948.8  336.41  4976.8  334.45  4988.1  331.19
  4990.9  330.69  4994.1  331.19  5005.4  332.45  5013.3  335.45  5098.3  336.51
  5121.3  335.99  5144.3   332.8  5156.6  334.74  5180.2  336.15  5215.6  335.62
  5284.3  337.43  5332.9  339.22    5534  341.62  5764.8  346.86  5970.3  351.29
#Mann= 9 ,-1 , 0
  3464.9      .1       0  3577.2     .05       0  4181.3     .16       0
  4340.7     .05       0  4876.7     .16       0  4988.1     .07       0
  4994.1     .16       0  5284.3     .05       0  5764.8     .16       0
Bank Sta=4948.8,5013.3
XS Rating Curve= 0 ,0
Exp/Cntr=0.3,0.1

Type RM Length L Ch R = 1 ,162240  ,1019,1019,1019
BEGIN DESCRIPTION:
Mapping XS 24a19fb8
END DESCRIPTION:
XS GIS Cut Line= 2
        3540960.     10278572.42      3539366.02     10277533.62
#Sta/Elev= 30
  3912.9   343.8    4107  340.16  4288.1     340  4417.8   339.2  4490.3  337.78
  4532.5  338.23  4547.6  337.54  4562.7  333.78  4577.8  332.86  4635.1  334.37
  4641.1  332.79  4692.5   333.9  4749.8  333.11  4764.9  334.37  4770.9  333.64
    4780  335.33    4786  334.58  4865.3  335.97  4936.9  334.34  4973.1  335.07
  4988.2   334.3  5000.3  331.83  5003.1  331.33  5006.3  331.83  5032.4  335.22
  5045.5  336.09  5169.3  336.84  5278.9  338.93  5414.1  342.24  5815.5  345.99
#Mann= 5 ,-1 , 0
  3912.9     .05       0  5000.3     .03       0  5006.3     .05       0
  5278.9     .16       0  5414.1     .05       0
Bank Sta=4988.2,5032.4
XS Rating Curve= 0 ,0
Exp/Cntr=0.3,0.1

Type RM Length L Ch R = 1 ,161221  ,294,294,294
BEGIN DESCRIPTION:
Mapping XS 6b78b523
END DESCRIPTION:
XS GIS Cut Line= 3
      3541324.54     10278021.17      3541042.43     10277825.87
      3539490.77     10277374.48
#Sta/Elev= 30
  4447.1   343.1  4512.4  342.23  4548.2   340.1  4577.9  340.46  4685.3  339.04
  4765.7  339.81  4905.1  334.68  4969.6  334.13  5006.3   329.3    5009   328.8
  5012.3   329.3  5019.7  331.38  5030.1  332.91  5364.4  334.44  5384.2  333.94
    5405  335.16  5570.7  334.72  5575.9  335.48  5609.5  332.63  5681.7  333.91
  5686.9  333.31  5715.2  334.02  5748.7  333.63  5759.2  334.64  5787.5  334.04
  5800.8  334.54  5893.3  339.27  6115.2  341.94  6269.4  342.59  6406.2   344.8
#Mann= 3 ,-1 , 0
  4447.1     .05       0  5006.3     .03       0  5012.3     .05       0
Bank Sta=4969.6,5030.1
XS Rating Curve= 0 ,0
Exp/Cntr=0.3,0.1

Type RM Length L Ch R = 1 ,160927  ,400,400,400
BEGIN DESCRIPTION:
WICKSON CREEK 108.0
END DESCRIPTION:
XS GIS Cut Line= 3
      3541442.15     10277741.66      3540846.56     10277490.68
      3539486.17     10277238.94
#Sta/Elev= 30
  4350.6  344.09  4359.8   344.8  4372.3  343.81  4388.9  339.62  4394.4  340.01
  4426.6  337.33  4542.2     336  4571.3  333.81  4618.8  335.98  4708.7  333.03
  4748.3  334.61  4908.2  332.36  4978.1  333.16  4990.9  331.88  4993.6   329.9
  4996.4   329.4  4999.6   329.9  5000.5   329.9  5017.9  332.21  5075.9  332.56
  5143.8  334.96  5297.7  333.71  5377.7  336.18  5448.9  336.23  5678.2  340.57
    5784  339.33  5894.8  340.65  6069.3   340.8  6232.6  343.96  6380.4  345.11
#Mann= 5 ,-1 , 0
  4350.6     .05       0  4908.2      .1       0  4993.6     .07       0
  4999.6      .1       0  5000.5     .05       0
Bank Sta=4978.1,5017.9
XS Rating Curve= 0 ,0
Exp/Cntr=0.3,0.1

Type RM Length L Ch R = 1 ,160527  ,968,968,968
BEGIN DESCRIPTION:
WICKSON CREEK 107.0
END DESCRIPTION:
XS GIS Cut Line= 3
      3541692.09     10277741.63      3540942.11     10277141.64
       3539492.1     10277041.64
#Sta/Elev= 30
  4065.8  345.74    4201  341.02  4221.9  341.84  4265.1  340.26  4300.3  342.97
  4335.5  339.94  4393.1  338.29  4500.4  337.23  4570.8  338.63  4734.1  336.07
  4841.4  331.89    4955  331.29  4995.2  328.94    4998  328.44  5001.2  328.94
  5028.8  329.34  5056.3  332.04  5136.5  330.91  5338.4  332.37  5406.1  333.48
  5587.6  334.38  5818.1  337.86  5918.4  335.86  6068.7  339.94  6219.1  342.15
  6239.1  339.99  6257.9  342.08  6262.9  341.21  6329.3  343.71  6479.7  345.56
#Mann= 5 ,-1 , 0
  4065.8     .05       0  4995.2     .03       0  5001.2     .05       0
  5338.4      .1       0  5406.1     .05       0
Bank Sta=4955,5056.3
XS Rating Curve= 0 ,0
Exp/Cntr=0.3,0.1

Type RM Length L Ch R = 1 ,159559  ,218,218,218
BEGIN DESCRIPTION:
WICKSON CREEK 106.0
END DESCRIPTION:
XS GIS Cut Line= 3
      3541842.08     10277641.62      3540642.11     10276441.64
      3539842.15     10276041.66
#Sta/Elev= 30
  3327.2  348.42  3496.9   343.7  3737.3  339.24  3793.9  338.88    3907  339.84
  4133.3  335.63  4409.3     334  4458.5  333.61  4505.8  334.43    4600  335.93
  4797.9  333.41  4882.8  334.27  4953.3  331.38  4981.8  331.01  5007.1  328.25
  5009.8  327.75  5013.1  328.25  5020.7  330.34  5032.6     331  5099.7  329.71
  5214.3  330.54    5382  330.74  5412.7  332.66  5440.7  335.62  5569.3  341.61
  5672.7  344.69  5843.2  345.55  5887.9  348.05  5904.7  350.75  5918.6  350.68
#Mann= 7 ,-1 , 0
  3327.2     .05       0  4409.3      .1       0  4505.8     .05       0
  4953.3      .1       0  5007.1     .07       0  5013.1      .1       0
  5214.3     .05       0
Bank Sta=4981.8,5032.6
XS Rating Curve= 0 ,0
Exp/Cntr=0.3,0.1

Type RM Length L Ch R = 1 ,159341  ,254,254,254
BEGIN DESCRIPTION:
WICKSON CREEK 105.0
END DESCRIPTION:
XS GIS Cut Line= 2
      3541869.74     10277429.92      3540014.25     10275498.48
#Sta/Elev= 30
  3399.2  346.46  3403.4  345.85  3438.6  344.62  3537.7  341.92  3827.6  337.91
  4450.2  334.09  4513.8  335.82    4627   335.3  4846.2  330.01  4888.6  330.32
  4909.7  329.74    4938  330.29  4980.5  329.73  4998.8  327.34  5001.6  326.84
  5004.8  327.34  5022.9  329.47  5065.4  329.15  5143.3  332.38    5221  333.68
  5369.5  333.92  5390.8  334.89  5468.5  335.07  5638.3  338.02  5744.3  339.05
  5765.7  340.36  5808.1  340.17  5857.5  341.72  5970.7  343.72  6077.5  346.63
#Mann= 3 ,-1 , 0
  3399.2     .05       0  4998.8     .03       0  5004.8     .05       0
Bank Sta=4980.5,5022.9
XS Rating Curve= 0 ,0
Exp/Cntr=0.3,0.1

Type RM Length L Ch R = 1 ,159087  ,572,572,572
BEGIN DESCRIPTION:
WICKSON CREEK 104.0
END DESCRIPTION:
XS GIS Cut Line= 2
       3541967.4     10277191.21      3540069.83     10275185.21
#Sta/Elev= 30
  3552.6  344.78  3662.1  341.67  3782.5  339.91  3888.5  339.59  3973.4  340.87
  4093.6  339.22  4242.1  338.98  4419.2  334.67  4532.1  333.92  4567.7  332.26
    4702  330.96    4808   331.7  4843.6  330.48  4963.7  329.78  5003.2  326.69
    5006  326.19  5009.2  326.69  5041.4   327.8  5062.9  329.89  5096.4  329.62
  5444.7  331.94  5536.6  335.74  5586.3  335.41  5786.1   338.8  5982.4  339.97
  6017.6  342.71  6053.2   343.7  6095.6  343.59  6291.8  348.06  6313.9   348.9
#Mann= 6 ,-1 , 0
  3552.6     .05       0  5003.2     .04       0  5009.2     .05       0
  5096.4     .05       0  5786.1     .08       0  6291.8     .05       0
Bank Sta=4963.7,5062.9
XS Rating Curve= 0 ,0
Exp/Cntr=0.3,0.1

Type RM Length L Ch R = 1 ,158515  ,496,496,496
BEGIN DESCRIPTION:
Mapping XS fbceb2e4
END DESCRIPTION:
XS GIS Cut Line= 2
      3542002.68     10276748.26      3540346.76     10275127.06
#Sta/Elev= 30
    3504  341.88  3947.5  336.48  4053.5  338.31  4166.7  337.35  4301.1  331.41
    4393  331.38  4428.4  329.56  4463.7  330.95  4605.8  331.09  4608.3  331.13
  4661.8  328.69  4817.3  329.52  4824.3  330.75  4838.5  328.83  4901.3  329.18
  4944.6  329.36  4972.9  327.03  4979.9  324.86  4998.2  324.35    5001  323.85
  5004.2  324.35  5008.2  327.47  5017.1  327.67  5043.7  329.43  5107.2   332.6
  5213.2  332.16  5496.1  335.27    5786  341.97  5807.3   340.9  5821.4  342.78
#Mann= 7 ,-1 , 0
    3504     .05       0  4605.8     .16       0  4608.3     .05       0
  4901.3     .16       0  4998.2     .07       0  5004.2     .16       0
  5017.1     .05       0
Bank Sta=4944.6,5043.7
XS Rating Curve= 0 ,0
Exp/Cntr=0.3,0.1

Type RM Length L Ch R = 1 ,158019  ,1021,1021,1021
BEGIN DESCRIPTION:
Mapping XS 511781c7
END DESCRIPTION:
XS GIS Cut Line= 2
       3541787.4     10276064.24      3540555.91     10274978.45
#Sta/Elev= 30
  4403.3  336.49  4522.2  336.88  4621.7  334.49  4650.2  335.05  4671.1  334.27
  4677.8   332.2    4692  331.57    4741  331.89  4844.6  332.17  4904.5  332.04
  4918.7  332.52  4926.3  334.18  4947.2  335.57  4961.4  334.73  4968.9  331.76
  4975.6  331.46  4983.2   327.2    4994  324.05  4996.7  323.55    5000  324.05
  5010.7  324.81  5018.3     327  5032.5  327.68    5153  328.62  5410.7  327.43
  5481.4  330.23  5537.9  330.67  5636.9  332.34  5891.9  336.06  6045.1  339.21
#Mann= 10 ,-1 , 0
  4403.3     .05       0    4741     .07       0  4844.6     .16       0
    4994     .07       0    5000     .16       0  5410.7     .05       0
  5481.4      .1       0  5537.9     .05       0  5636.9      .1       0
  5891.9     .05       0
#XS Ineff= 2 , 0
         4941.02  335.61
Permanent Ineff=
       F       F
Bank Sta=4975.6,5032.5
XS Rating Curve= 0 ,0
Exp/Cntr=0.3,0.1

Type RM Length L Ch R = 1 ,156998  ,239,239,239
BEGIN DESCRIPTION:
WICKSON CREEK 103.0
END DESCRIPTION:
XS GIS Cut Line= 4
      3542342.11     10276541.65      3542015.99     10275576.59
       3540896.2     10274790.14      3540156.85     10274467.32
#Sta/Elev= 30
  3458.1  344.63  3788.4   340.4  3851.3  338.44  4526.6  332.01    4598  331.48
  4612.9  332.23  4812.4  329.42  4892.6  328.99  4950.8  329.89    4964   329.5
  4996.8  323.25  4999.5  322.75  5002.8  323.25  5014.6  324.79  5035.5  324.31
  5050.3  325.92  5142.7  326.51  5172.3  327.85  5270.4  327.58  5395.4  331.93
  5594.9  332.63  5776.2  335.16  5854.5  334.84    5977  337.61  6035.1  340.64
  6067.8  339.92  6151.7  342.41  6209.7  342.83  6256.3  344.85  6651.9  350.67
#Mann= 5 ,-1 , 0
  3458.1     .05       0  4950.8     .16       0  4996.8     .07       0
  5002.8     .16       0  5270.4     .05       0
Bank Sta=4964,5014.6
XS Rating Curve= 0 ,0
Exp/Cntr=0.3,0.1

Type RM Length L Ch R = 1 ,156759  ,915,915,915
BEGIN DESCRIPTION:
WICKSON CREEK 101.0
END DESCRIPTION:
XS GIS Cut Line= 3
       3542392.1     10275591.64      3541592.11     10275041.64
      3540792.13     10274341.67
#Sta/Elev= 30
    4027  343.03  4192.8  336.89  4378.9  332.35  4530.3  330.84  4616.9  328.68
  4765.3   327.9  4826.4  327.92  4897.7  326.83  4918.7  324.17  4939.6  324.27
  4948.5  325.31  4975.5  325.03  4991.8  322.68  4994.5  322.18  4997.8  322.68
  5019.2  325.38  5046.9  325.41  5054.3  325.64  5076.1  329.28  5082.8  329.45
  5295.4  329.89  5458.6  332.91  5571.6  332.66  5784.2  336.27  5826.9  338.52
  5855.4   337.6  5883.8   339.6  5990.1   341.1  6032.8  343.33  6060.8  343.87
#Mann= 6 ,-1 , 0
    4027     .05       0  4765.3      .1       0  4826.4     .16       0
  4991.8     .07       0  4997.8     .16       0  5046.9     .05       0
Bank Sta=4975.5,5019.2
XS Rating Curve= 0 ,0
Exp/Cntr=0.3,0.1

Type RM Length L Ch R = 1 ,155844  ,708,708,708
BEGIN DESCRIPTION:
WICKSON CREEK 99.0
END DESCRIPTION:
XS GIS Cut Line= 2
      3542931.29      10275402.3      3540918.41     10273805.88
#Sta/Elev= 30
  3405.3  336.29  3526.3   336.7  3931.7  334.65  4173.6   335.2  4237.7  334.42
  4330.6  329.87  4611.9  327.91  4657.5  326.68  4741.5  326.82  4942.7  324.07
    4978  324.61  4996.7  320.95  4999.4  320.45  5002.7  320.95  5006.8  323.04
  5013.2  323.17  5021.3   324.8  5070.4  327.49  5362.5  331.92  5397.8  333.06
  5420.2  335.82  5455.5  334.04  5469.9  335.92  5668.6  338.66  5697.4  340.37
  5718.2  339.56  5753.5  341.07  5825.6  341.37  5939.4  344.52  5974.4  344.52
#Mann= 6 ,-1 , 0
  3405.3     .05       0  4611.9      .1       0  4741.5     .16       0
  4996.7     .07       0  5002.7     .16       0  5070.4     .05       0
Bank Sta=4978,5021.3
XS Rating Curve= 0 ,0
Exp/Cntr=0.3,0.1

Type RM Length L Ch R = 1 ,155136  ,1390,1390,1390
BEGIN DESCRIPTION:
WICKSON CREEK 98.0
END DESCRIPTION:
XS GIS Cut Line= 3
      3543692.11     10275541.64       3541843.7     10273832.45
       3540982.6     10273603.29
#Sta/Elev= 30
    3035  337.61  3827.4  333.19  4273.6  331.91  4605.9  332.43  4782.8  331.12
  4931.4  328.11  4947.6  325.95  4981.2  323.16  4999.2  320.03    5002  319.53
  5005.2  320.03  5023.5  323.27  5227.1  325.51  5441.1  326.74  5469.4  325.49
  5476.2  326.56  5483.6  325.06  5497.8  324.77  5564.5  324.93  5585.2  328.69
  5612.6  325.55  5637.9   325.8    5668  326.96  5692.8  325.67  5713.8  327.16
  5823.2  333.39    5875  338.37    5906  336.36  5928.5  337.65  6443.6  344.99
#Mann= 8 ,-1 , 0
    3035     .05       0  4947.6     .16       0  4999.2     .07       0
  5005.2     .16       0  5227.1     .05       0  5612.6      .1       0
  5637.9     .16       0  5713.8     .05       0
Bank Sta=4931.4,5023.5
XS Rating Curve= 0 ,0
Exp/Cntr=0.3,0.1

Type RM Length L Ch R = 1 ,153746  ,1132,1132,1132
BEGIN DESCRIPTION:
Mapping XS f7e3e313
END DESCRIPTION:
XS GIS Cut Line= 3
      3543569.29     10274430.89      3541837.56     10273144.46
      3541360.95     10273079.35
#Sta/Elev= 30
  3144.1  331.14  3591.3  330.84  3756.1  332.33  4099.8   332.6  4463.3  328.96
  4571.8  326.93  4670.2  323.62  4677.4  323.59  4713.6  325.64  4757.4  326.26
  4957.7  324.25  4984.8  320.33  4996.4  317.76  4999.2  317.26  5002.4  317.76
    5014  322.69  5028.6  323.27  5071.5  322.07  5101.2  323.19    5135  322.41
  5170.6  323.58  5243.5  330.09  5285.2  332.31  5355.7  337.46  5367.4  336.88
  5438.1  340.11  5549.1  342.47    5718  343.88  5760.8  344.36  5782.4  344.71
#Mann= 9 ,-1 , 0
  3144.1     .05       0  4670.2     .16       0  4677.4     .05       0
  4996.4    .035       0  5002.4     .05       0  5101.2      .1       0
  5170.6     .05       0    5718      .1       0  5760.8     .05       0
Bank Sta=4957.7,5014
XS Rating Curve= 0 ,0
Exp/Cntr=0.3,0.1

Type RM Length L Ch R = 1 ,152614  ,897,897,897
BEGIN DESCRIPTION:
WICKSON CREEK 96.0
END DESCRIPTION:
XS GIS Cut Line= 4
      3544892.12     10275191.67      3543378.42     10273061.62
      3541982.24     10272660.06      3541336.91     10272908.78
#Sta/Elev= 30
  1590.5  342.19  2007.5  336.52  2803.2  332.17  2950.6  331.59  3448.1  327.76
    3559  328.08  3663.8  326.31  3691.2  323.35  3741.7  326.72  3842.5  328.97
  4100.8  327.58  4441.5  330.04  4813.7  325.92    4833   324.9  4844.9  322.36
  4897.2  320.92  4969.8  319.85  4983.4  318.79    4998  314.61  5000.8  314.11
    5004  314.61  5022.3  319.85  5068.6  322.44  5089.7  323.34  5346.4  327.22
  5506.8  327.63  5735.3  332.06  5813.8  334.17  6188.4   341.5    6348  343.89
#Mann= 13 ,-1 , 0
  1590.5     .05       0  2803.2      .1       0  2950.6     .05       0
  3448.1      .1       0    3559     .05       0  4897.2     .16       0
    4998     .07       0    5004     .16       0  5068.6      .1       0
  5506.8     .05       0  5735.3      .1       0  5813.8     .05       0
  6188.4      .1       0
#XS Ineff= 2 , 0
         3856.82  329.06
Permanent Ineff=
       F       F
Bank Sta=4969.8,5089.7
XS Rating Curve= 0 ,0
Exp/Cntr=0.3,0.1

Type RM Length L Ch R = 1 ,151717  ,1674,1674,1674
BEGIN DESCRIPTION:
WICKSON CREEK 95.0
END DESCRIPTION:
XS GIS Cut Line= 4
      3545690.91     10274790.78      3543246.48     10272367.18
      3542100.64     10272096.34      3541156.61     10272519.77
#Sta/Elev= 30
  1084.6  344.65  1139.7  345.02  1203.4  340.85  1995.3  335.15  3536.8  327.93
  3642.9  323.28  3713.6   324.9  3741.9  321.59  3763.1   323.6  3918.7  328.13
  4073.2  327.02  4132.2  326.99  4369.4  326.56  4456.1  327.59  4550.3  324.73
  4800.3  323.68  4925.1  321.32  4952.6  319.99  5000.1   313.1  5002.9   312.6
  5006.1   313.1  5014.3   317.2  5045.1  318.93    5151  320.61  5272.3  320.89
  5484.5  327.32  6001.1  331.14  6272.6  338.88  6616.7  343.16  6738.9  344.38
#Mann= 12 ,-1 , 0
  1084.6     .05       0  4073.2      .1       0  4132.2     .05       0
  4369.4      .1       0  4550.3     .16       0  4800.3      .1       0
  4925.1     .16       0  5000.1     .07       0  5006.1     .16       0
    5151      .1       0  5484.5     .05       0  6616.7      .1       0
#XS Ineff= 2 , 0
         3928.41  328.07
Permanent Ineff=
       F       F
Bank Sta=4952.6,5045.1
XS Rating Curve= 0 ,0
Exp/Cntr=0.3,0.1

Type RM Length L Ch R = 1 ,150043  ,1047,1047,1047
BEGIN DESCRIPTION:
WICKSON CREEK 93.0
END DESCRIPTION:
XS GIS Cut Line= 3
      3545975.66     10274311.64      3542711.75      10271401.9
      3541329.77     10271846.35
#Sta/Elev= 30
  1441.4  345.38  1911.6  342.35  2577.1  332.48  3894.7  326.32  3993.4   319.6
  4043.6  323.76  4227.5  326.26  4588.6  326.49  4659.7  326.53  4725.6  323.14
  4801.1  319.94  4949.9  320.43  4970.8  317.76  4978.3   314.2    4985  314.64
  4992.5  311.06  5010.4  310.46  5013.2  309.96  5016.4  310.46  5049.4  316.41
    5077  317.37  5227.6  319.39  5460.6  323.14  5473.5  323.85    5611  323.92
  5674.6  323.91  5857.2  326.41    6251  325.79  6813.1  331.25  7265.7  339.42
#Mann= 12 ,-1 , 0
  1441.4     .05       0  4588.6      .1       0  4725.6     .16       0
  5010.4     .07       0  5016.4     .16       0  5227.6     .05       0
  5460.6      .1       0  5473.5     .05       0    5611      .1       0
  5674.6     .05       0  5857.2      .1       0    6251     .05       0
#XS Ineff= 2 , 0
         4221.59  326.29
Permanent Ineff=
       F       F
Bank Sta=4949.9,5077
XS Rating Curve= 0 ,0
Exp/Cntr=0.3,0.1

Type RM Length L Ch R = 1 ,148996  ,677,677,677
BEGIN DESCRIPTION:
WICKSON CREEK 92.0
END DESCRIPTION:
XS GIS Cut Line= 3
      3545392.09     10272391.63      3542552.03     10270915.79
      3541192.07     10271491.66
#Sta/Elev= 30
  3028.1  333.47  3345.9  327.71  3489.4  321.55  3533.6  321.97  3583.5  318.14
  3644.2  323.57    3689  323.62  3718.1  323.39  4058.7   325.8  4151.6   323.2
  4245.2   319.3  4257.7  315.83  4296.3   321.4  4392.9  322.17    4733   325.4
  4843.8  322.77  4970.6  317.39  4997.3  308.72    5000  308.22  5003.3  308.72
  5014.8  311.86  5081.1  315.78  5268.9  318.01  5369.7     322  5385.1  325.29
  5417.2  321.88  5981.4  324.58  6151.1   324.5  6949.9  327.83  7705.6  339.69
#Mann= 11 ,-1 , 0
  3028.1     .05       0    3689      .1       0  3718.1     .05       0
  4151.6     .16       0  4392.9     .05       0  4843.8     .16       0
  4997.3     .07       0  5003.3     .16       0  5369.7     .05       0
  5981.4      .1       0  6151.1     .05       0
#XS Ineff= 2 , 0
          4735.8   325.5
Permanent Ineff=
       F       F
Bank Sta=4997.3,5003.3
XS Rating Curve= 0 ,0
Exp/Cntr=0.3,0.1

Type RM Length L Ch R = 1 ,148319  ,537,537,537
BEGIN DESCRIPTION:
Mapping XS 09543423
END DESCRIPTION:
XS GIS Cut Line= 2
      3545635.16     10272175.55      3543132.96     10270693.26
#Sta/Elev= 30
  2549.9  332.67  3207.4  323.65  3233.9  321.73  3239.7  319.29  3276.8  316.76
    3308  319.02  3430.8  318.87  3467.9  321.69  3574.7  322.52  3680.4  324.63
    3933  318.82  3940.4   318.8  4000.1  317.36  4021.5  313.96  4037.1  318.47
  4074.2  320.94  4181.4  323.91  4271.1  324.63  4651.2  317.14  4729.2  315.59
  4898.8  318.18  4984.6  312.88  4994.3  310.51  4997.2   306.9  4999.9   306.4
  5003.2   306.9  5024.8  316.22  5037.2  319.08  5181.5  322.23  5458.2  322.17
#Mann= 9 ,-1 , 0
  2549.9     .05       0  3207.4      .1       0  3574.7     .05       0
    3933     .16       0  3940.4     .05       0  4651.2     .16       0
  4997.2     .07       0  5003.2     .16       0  5024.8     .05       0
#XS Ineff= 2 , 0
         4271.02  324.71
Permanent Ineff=
       F       F
Bank Sta=4984.6,5037.2
XS Rating Curve= 0 ,0
Exp/Cntr=0.3,0.1

Type RM Length L Ch R = 1 ,147782  ,846,846,846
BEGIN DESCRIPTION:
Mapping XS e02ddf3c
END DESCRIPTION:
XS GIS Cut Line= 3
       3545382.1      10271573.7      3544080.27     10270854.04
      3543460.63     10270416.41
#Sta/Elev= 30
  3417.3   325.9  3742.4   324.9  3845.5  322.89  3883.3  320.47    3889  321.79
  3926.9  317.28  3970.4  320.52  4026.9  318.75  4102.9  316.97  4148.6  312.22
  4170.8  315.84  4290.5   318.7  4460.9  320.65  4565.7  322.94  4670.8  322.99
  4898.2   322.4    4955  321.15  4969.8  318.49  4984.5  310.84  4990.7  311.42
  4996.3  308.24  5002.5  306.11  5005.2  305.61  5008.5  306.11  5012.7  312.76
  5171.7  318.69  5322.3  318.28  5457.3   317.3  5537.4  320.15  5663.4  320.37
#Mann= 10 ,-1 , 0
  3417.3     .05       0  4026.9     .12       0  4290.5     .16       0
  4460.9      .1       0  4565.7     .05       0  4670.8      .1       0
  4996.3     .16       0  5002.5     .07       0  5008.5     .16       0
  5322.3     .05       0
#XS Ineff= 2 , 0
         4588.64  323.65
Permanent Ineff=
       F       F
Bank Sta=4969.8,5012.7
XS Rating Curve= 0 ,0
Exp/Cntr=0.3,0.1

Type RM Length L Ch R = 1 ,147044  ,1591,1591,1591
BEGIN DESCRIPTION:
Mapping XS 1dce0ea9
END DESCRIPTION:
XS GIS Cut Line= 2
      3545396.02     10271067.66      3543572.25     10269753.54
#Sta/Elev= 30
  3490.4  326.99  3712.7  329.83  3885.3  329.07  3976.6   327.7  4091.9  318.48
  4121.4  318.15  4142.2  314.93    4157  316.29  4164.7  315.02  4271.7  312.97
  4299.3   310.7    4314  311.49    4321  313.52  4388.9  315.83  4493.6  317.98
  4607.4  314.68  4844.2  316.58  4959.5  314.77  4995.1  307.43  4998.3  304.39
    5001  303.89  5004.3  304.39  5009.8  307.14    5016  312.36  5036.9   314.9
  5084.6  316.13  5101.9   317.9  5231.9   320.8  5525.3  319.03  5738.3  320.66
#Mann= 7 ,-1 , 0
  3490.4     .05       0  3885.3      .1       0  4164.7     .12       0
  4388.9     .16       0  4998.3     .07       0  5004.3     .16       0
  5084.6     .05       0
Bank Sta=4959.5,5036.9
XS Rating Curve= 0 ,0
Exp/Cntr=0.3,0.1

Type RM Length L Ch R = 1 ,145453  ,1793,1793,1793
BEGIN DESCRIPTION:
WICKSON CREEK 91.0
END DESCRIPTION:
XS GIS Cut Line= 4
      3545978.63     10270982.05      3545395.47     10270126.72
       3544223.6     10269399.73      3543476.01     10269648.92
#Sta/Elev= 30
  3711.3  325.27  4018.1  323.17  4083.9  321.88  4125.8  319.42  4186.7  321.51
    4401  323.22  4586.6  323.38  4694.8  321.73  4819.7  318.37  4903.9  312.39
  4971.2  310.77  4985.8  309.37  4995.4  303.98  4998.1  303.48  5001.4  303.98
  5013.7  305.69  5021.1  310.41    5035  313.84  5239.4  314.64  5297.2   313.5
  5456.6   316.7  5480.1  315.73  5549.2  316.27  5549.9  316.27  5638.6  315.35
  6009.6  316.75  6095.7  318.46    6277  317.92    6359  319.63  6913.6  320.55
#Mann= 9 ,-1 , 0
  3711.3     .05       0  4186.7      .1       0    4401     .16       0
  4694.8      .1       0  4819.7     .16       0  4995.4     .07       0
  5001.4     .16       0  5549.2      .1       0  5549.9     .05       0
Bank Sta=4971.2,5035
XS Rating Curve= 0 ,0
Exp/Cntr=0.3,0.1

Type RM Length L Ch R = 1 ,143660  ,133,133,133
BEGIN DESCRIPTION:
WICKSON CREEK 90.0
END DESCRIPTION:
XS GIS Cut Line= 6
      3546384.93     10268903.96      3545421.36     10269023.76
      3545119.28     10269148.76      3544817.19     10269252.92
      3544577.61     10269252.92      3543886.03     10269206.13
#Sta/Elev= 30
  3591.2  334.35    3725  327.16  3966.9  319.04  4299.3  314.87  4592.2  312.03
  4650.8  313.46  4669.3  310.37  4674.7  311.61  4691.2  306.97    4704  306.05
  4727.9  310.43  4900.1  310.65  4918.2  310.51  4960.2  307.77  4970.1  305.39
  4975.3  306.47  4991.9  301.15    5001  301.33  5003.5  300.76  5006.3  300.26
  5009.5  300.76  5037.7   310.1    5195  315.17  5323.7  316.13  5383.7  314.95
  5448.2  315.16  5689.3  317.97  5838.6  317.18  5954.9  318.48  6141.4  318.52
#Mann= 7 ,-1 , 0
  3591.2     .05       0  4299.3      .1       0  4900.1     .16       0
    5001      .1       0  5003.5     .07       0  5009.5      .1       0
    5195     .05       0
Bank Sta=4918.2,5037.7
XS Rating Curve= 0 ,0
Exp/Cntr=0.3,0.1

Type RM Length L Ch R = 1 ,143527  ,944,944,944
BEGIN DESCRIPTION:
Mapping XS f6fca8eb
END DESCRIPTION:
XS GIS Cut Line= 4
      3546416.12     10268784.18      3545369.28     10268898.76
      3544801.57     10269159.17      3543900.49     10269127.92
#Sta/Elev= 30
  3572.5  333.05  3775.8  325.19  4039.3  318.02  4170.1  315.43  4459.8  313.36
  4542.3  312.96  4633.5  310.59  4687.7  312.36  4754.5  313.01  4798.5  310.38
  4882.7  308.64  4951.7  309.96  4974.5  308.31  4980.2  305.77  4985.7  301.85
  4993.5  299.72  4996.3  299.22  4999.5  299.72  5026.2  307.82  5049.1  310.48
  5214.3  313.74  5339.7   315.8  5459.8  315.14  5649.9  317.48    5810  317.06
    5870  318.34  5897.6  317.48  5902.6  318.27  6030.1   318.9  6151.8  318.26
#Mann= 5 ,-1 , 0
  3572.5     .05       0  4459.8      .1       0  4993.5     .07       0
  4999.5      .1       0  5214.3     .05       0
Bank Sta=4951.7,5049.1
XS Rating Curve= 0 ,0
Exp/Cntr=0.3,0.1

Type RM Length L Ch R = 1 ,142583  ,2731,2731,2731
BEGIN DESCRIPTION:
WICKSON CREEK 88.0
END DESCRIPTION:
XS GIS Cut Line= 3
      3546239.58     10268672.75      3544878.42     10268228.29
      3542670.13     10269040.77
#Sta/Elev= 30
  3824.2  325.04  4273.9  314.81  4412.2  313.75  4541.6  313.33  4736.7  312.35
  4810.5  309.78    4884  307.74  4972.4   308.9  4989.2   303.9  5001.3  297.79
  5004.1  297.29  5007.3  297.79  5010.3  301.44  5020.8  305.54    5031  306.94
  5073.4  308.06  5094.4  306.74  5134.2  309.07  5358.7  315.02  5635.8  315.97
  5709.9  314.33  5892.6   317.7    6029  315.74  6451.6  318.16  6611.2  318.89
  6652.8  319.01  6759.6  319.56  7163.8  321.62  7391.5  319.69  7609.1  320.31
#Mann= 11 ,-1 , 0
  3824.2     .05       0  4412.2      .1       0  4541.6     .05       0
  4810.5     .16       0  5001.3     .07       0  5007.3     .16       0
  5134.2     .05       0  6451.6      .1       0  6611.2     .05       0
  6652.8      .1       0  6759.6     .05       0
Bank Sta=4972.4,5031
XS Rating Curve= 0 ,0
Exp/Cntr=0.3,0.1

Type RM Length L Ch R = 1 ,139852  ,1013,1013,1013
BEGIN DESCRIPTION:
WICKSON CREEK 87.0
END DESCRIPTION:
XS GIS Cut Line= 4
      3545857.36     10267741.58      3545399.25     10267249.12
      3544795.09     10267013.01      3544526.98      10267030.1
#Sta/Elev= 30
  3947.2  315.24  4056.8  313.04  4205.8  311.27  4417.9  313.27    4517  312.85
  4583.8  311.68  4614.7  311.62  4685.4  310.99  4745.6  306.68  4863.7  305.23
  4917.3   303.7  4949.6  301.88    4971  303.58  4980.1  300.62  4985.4  297.36
  4992.5  294.81  5009.9  294.12  5012.3  293.28    5015  292.78  5018.3  293.28
  5034.4  295.23  5039.8  296.66  5046.2  299.43  5064.2  303.79  5069.6  302.16
  5088.7   306.7  5164.2   309.3  5321.1  311.88  5484.8  316.01  5537.1  315.82
#Mann= 7 ,-1 , 0
  3947.2     .05       0  4583.8     .16       0  4614.7     .05       0
  4685.4     .16       0  5012.3     .07       0  5018.3     .16       0
  5164.2     .05       0
Bank Sta=4971,5064.2
XS Rating Curve= 0 ,0
Exp/Cntr=0.3,0.1

Type RM Length L Ch R = 1 ,138839  ,2531,2531,2531
BEGIN DESCRIPTION:
WICKSON CREEK 86.0
END DESCRIPTION:
XS GIS Cut Line= 4
      3546302.84     10266959.28      3545725.64     10266443.56
      3544454.81     10266158.84      3544292.72     10266189.34
#Sta/Elev= 30
  3853.3  310.22  4053.5   309.5  4072.6  309.67  4227.8  308.64  4236.7  308.63
  4366.8  308.86  4376.1  307.93    4461  306.33  4631.7  310.05  4733.4  307.62
  4798.1     303  4943.3   303.5  4948.6   303.3  4969.1  302.13  4989.6  294.34
  4996.9  293.89  4999.6  293.39  5002.9  293.89  5020.1  297.44  5030.6  303.07
  5051.1  305.17  5282.7  306.06  5409.8  309.53  5648.6  309.09  5668.2  309.01
  5696.7  305.95    5748  306.21  5778.7  309.32  5813.6  308.41  6094.6  315.03
#Mann= 13 ,-1 , 0
  3853.3     .05       0  4053.5      .1       0  4072.6     .05       0
  4227.8      .1       0  4236.7     .05       0  4366.8      .1       0
  4376.1     .05       0  4943.3     .16       0  4996.9     .07       0
  5002.9     .16       0  5282.7     .05       0  5648.6     .16       0
  5813.6     .05       0
Bank Sta=4948.6,5051.1
XS Rating Curve= 0 ,0
Exp/Cntr=0.3,0.1

Type RM Length L Ch R = 1 ,136308  ,873,873,873
XS GIS Cut Line= 2
      3547078.24    10266146.389     3545414.177    10265086.493
#Sta/Elev= 30
       0   307.1   39.96  307.31   69.93   306.5  459.52  306.45  499.48  307.22
  529.45  306.97  739.23  308.38   769.2  307.77  869.09  302.96  909.05  303.22
  939.02  304.19 1008.95  303.84 1078.87  302.18 1258.69  302.07 1328.61  301.52
 1358.58  300.68 1388.55  301.53 1428.51  300.95 1488.45  301.22 1498.44  300.89
 1508.42  298.52 1518.41  295.21  1528.4  293.52 1538.39   293.9 1548.38  296.57
 1558.37  302.01 1568.36  305.77 1578.35  307.02 1618.31  308.01 1977.93  309.69
#Mann= 3 ,-1 , 0
       0     .05       0 1488.45     .07       0 1558.37     .05       0
Bank Sta=1498.44,1558.37
XS Rating Curve= 0 ,0
Exp/Cntr=0.3,0.1

Type RM Length L Ch R = 1 ,135435  ,1023,1023,1023
BEGIN DESCRIPTION:
WICKSON CREEK 84.0
END DESCRIPTION:
XS GIS Cut Line= 4
      3547483.05     10265950.71       3547219.1     10265136.06
      3545732.56     10264723.73      3545398.17     10264833.32
#Sta/Elev= 30
  3276.4  311.11  3554.6  304.71  4390.8  303.94  4472.3  302.27  4492.2  299.59
    4524  298.32  4555.1  300.86  4619.8  298.74  4659.2  291.61  4688.3  298.31
  4742.2  300.03  4897.7   299.8    4949  301.17  4970.2  298.64  4985.4  290.78
  4988.2  290.28  4991.4  290.78  5001.3  293.55  5011.7  299.67  5022.1  300.94
  5067.4  300.29  5100.4  303.39  5201.8  302.78  5260.8  303.61  5303.1  301.31
    5328  298.49  5519.2  305.28  5632.5   305.9  5703.6  306.67  6027.3  310.48
#Mann= 13 ,-1 , 0
  3276.4     .05       0  4390.8     .16       0  4492.2     .12       0
  4742.2     .05       0  4897.7     .16       0  4985.4     .07       0
  4991.4     .16       0  5100.4      .1       0  5201.8     .05       0
  5303.1      .1       0  5519.2     .05       0  5632.5      .1       0
  5703.6     .05       0
Bank Sta=4949,5022.1
XS Rating Curve= 0 ,0
Exp/Cntr=0.3,0.1

Type RM Length L Ch R = 1 ,134412  ,1594,1594,1594
BEGIN DESCRIPTION:
Mapping XS 6d187f69
END DESCRIPTION:
XS GIS Cut Line= 4
      3547098.86     10264700.89      3546896.22     10264393.65
      3546147.52     10264057.28      3545701.93     10264172.16
#Sta/Elev= 30
  4154.8  307.93  4318.5  307.14    4565  304.67  4604.1  302.87    4627   300.5
  4680.8  296.72  4732.7  298.07    4779  298.36  4804.5  297.69  4946.1  298.25
  4957.6  297.93  4980.7  296.39  4987.8  291.33  4995.4  288.31  4998.2  287.81
  5001.4  288.31  5003.9  288.56  5009.7  295.97  5027.1  298.76  5032.6  298.62
  5052.5  300.59  5067.3  301.22  5171.5  302.47  5246.5  301.86  5298.3  300.32
  5305.7  301.42  5423.9  302.36  5514.5  304.76  5657.7  305.53  5803.8  307.92
#Mann= 8 ,-1 , 0
  4154.8     .05       0    4627     .16       0  4804.5     .05       0
  4946.1     .12       0  4995.4     .07       0  5001.4     .12       0
  5052.5     .16       0  5067.3     .05       0
Bank Sta=4957.6,5027.1
XS Rating Curve= 0 ,0
Exp/Cntr=0.3,0.1

Type RM Length L Ch R = 1 ,132818  ,2100,2100,2100
BEGIN DESCRIPTION:
WICKSON CREEK 83.0
END DESCRIPTION:
XS GIS Cut Line= 4
      3547446.76     10264347.15      3547373.65     10263927.07
       3546765.2     10263205.62      3546496.86     10263125.53
#Sta/Elev= 30
  3734.7  305.61  3994.1  307.08  4032.8  306.14  4065.4  305.95  4415.1  295.12
  4444.3  296.17  4545.5  297.16  4691.8  295.99  4710.1  296.06  4838.1  295.93
  4843.1  296.12  4946.7  295.95    4961   294.5  4967.5  290.05  4975.3  291.54
  4981.8  287.77  4993.1  287.64  4995.9  287.14  4999.1  287.64  5003.9  287.66
  5010.4  291.02  5018.2  289.97  5024.7  292.88  5045.5  297.75  5053.3   303.3
  5074.1  310.28    5117  311.71  5122.9   311.9  5295.9  314.19  5384.9  313.73
#Mann= 14 ,-1 , 0
  3734.7     .05       0  4032.8      .1       0  4065.4     .05       0
  4415.1     .16       0  4444.3     .05       0  4545.5     .16       0
  4691.8     .12       0  4710.1     .16       0  4838.1     .12       0
  4843.1     .16       0  4993.1     .07       0  4999.1     .16       0
    5117      .1       0  5122.9     .05       0
Bank Sta=4946.7,5045.5
XS Rating Curve= 0 ,0
Exp/Cntr=0.3,0.1

Type RM Length L Ch R = 1 ,130718  ,1381,1381,1381
BEGIN DESCRIPTION:
WICKSON CREEK 82.0
END DESCRIPTION:
XS GIS Cut Line= 4
      3548371.91     10265185.79      3548232.46     10263585.03
      3548299.37     10262403.75      3548122.34     10261648.42
#Sta/Elev= 30
    2609   314.2  2673.4     312    2892  310.83  3175.3  304.72  3506.5  300.03
  3797.6   299.6  4018.5  295.09  4118.8  298.93    4220  297.38  4319.4  291.51
  4449.6  296.76  4619.9  297.81  4810.2  291.43  4960.4  294.23  4970.4  292.99
  4990.5  286.85  5007.5   285.4  5010.2   284.9  5013.5   285.4  5050.6  293.44
  5100.6   294.9  5183.9  291.41    5311  293.11  5357.5  298.63  5362.5  297.84
  5402.6  301.94  5462.8  309.88  5720.2  326.91  5863.4  333.14  6174.8   334.4
#Mann= 3 ,-1 , 0
    2609     .05       0  5007.5    .035       0  5013.5     .05       0
Bank Sta=4960.4,5050.6
XS Rating Curve= 0 ,0
Exp/Cntr=0.3,0.1

Type RM Length L Ch R = 1 ,129337  ,864,864,864
BEGIN DESCRIPTION:
WICKSON CREEK 81.0
END DESCRIPTION:
XS GIS Cut Line= 3
      3550642.13     10264841.68      3549242.11     10262441.64
      3548592.11     10261691.65
#Sta/Elev= 30
  2206.4  335.12  2331.7  331.65  2636.9  319.03  3075.1  309.07  3699.5   304.8
  3801.2  304.46  3873.5  305.74  3977.3  303.55  4415.6  304.93  4752.2  295.78
  4800.9  297.75    4846  296.92  4881.2  292.37  4955.6  290.59  4971.3  291.86
  4977.1  286.74  4984.7  285.49  4995.7  283.67  4998.4  283.17  5001.7  283.67
  5012.9  288.21  5019.7  289.36  5034.8  291.28  5077.6   291.3  5233.3  295.56
  5431.8  297.51  5594.2  302.23  5736.7  311.93  5849.7   322.4  5977.4  329.32
#Mann= 5 ,-1 , 0
  2206.4     .05       0  4984.7      .1       0  4995.7     .07       0
  5001.7      .1       0  5019.7     .05       0
Bank Sta=4971.3,5034.8
XS Rating Curve= 0 ,0
Exp/Cntr=0.3,0.1
